--- CAMPGROUND CREEK.prj (project) ---

Proj Title=CAMPGROUND CREEK Base Level Engineering
Current Plan=p01
Default Exp/Contr=0.3,0.1
English Units
Geom File=g01
Flow File=f01
Plan File=p01
Y Axis Title=Elevation
X Axis Title(PF)=Main Channel Distance
X Axis Title(XS)=Station
BEGIN DESCRIPTION:
CAMPGROUND CREEK
END DESCRIPTION:
DSS Export Rating Curves= 0
DSS Export Rating Curve Sorted= 0
DSS Export Volume Flow Curves= 0
DXF OffsetX= 0
DXF OffsetY= 0
DXF ScaleX= 1
DXF ScaleY= 10

--- CAMPGROUND CREEK.p01 (plan) ---

Plan Title=Multiple Run
Short Identifier=Multiple
Geom File=g01
Flow File=f01
Subcritical Flow
K Sum by GR= 0
Std Step Tol= 0.01
Critical Tol= 0.01
Num of Std Step Trials= 20
Max Error Tol= 0.3
Flow Tol Ratio= 0.001
Split Flow NTrial= 30
Split Flow Tol= 0.02
Split Flow Ratio= 0.02
Log Output Level= 0
Friction Slope Method= 1
Unsteady Friction Slope Method= 2
Unsteady Bridges Friction Slope Method= 1
Parabolic Critical Depth
Global Vel Dist=  1 , 1 , 1
Global Log Level= 0
CheckData=True
Encroach Param= -1, 0, 0, 0
BEGIN DESCRIPTION:
Multiple Run
END DESCRIPTION:

--- CAMPGROUND CREEK.f01 (steady flow) ---

Flow Title=Multiple
Number of Profiles=7
Profile Names=10-year,25-year,50-year,1pct_min,100-year,1pct_plu,500-year
River Rch & RM= CAMPGROUND CREEK,Reach-1,47500
     490     803    1109     798    1495    2800    2078
River Rch & RM= CAMPGROUND CREEK,Reach-1,36163
     746    1255    1670    1168    2264    4391    3104
River Rch & RM= CAMPGROUND CREEK,Reach-1,31513
    1077    1860    2150    1415    2900    5945    3899
River Rch & RM= CAMPGROUND CREEK,Reach-1,24500
    1374    2425    2631    1651    3559    7673    4767
River Rch & RM= CAMPGROUND CREEK,Reach-1,15500
    1750    3125    3628    2307    4966   10690    6644
Boundary for River Rch & Prof#=CAMPGROUND CREEK,Reach-1,1
Up Type=0
Dn Type=3
Dn Slope=0.005
Boundary for River Rch & Prof#=CAMPGROUND CREEK,Reach-1,2
Up Type=0
Dn Type=3
Dn Slope=0.005
Boundary for River Rch & Prof#=CAMPGROUND CREEK,Reach-1,3
Up Type=0
Dn Type=3
Dn Slope=0.005
Boundary for River Rch & Prof#=CAMPGROUND CREEK,Reach-1,4
Up Type=0
Dn Type=3
Dn Slope=0.005
Boundary for River Rch & Prof#=CAMPGROUND CREEK,Reach-1,5
Up Type=0
Dn Type=3
Dn Slope=0.005
Boundary for River Rch & Prof#=CAMPGROUND CREEK,Reach-1,6
Up Type=0
Dn Type=3
Dn Slope=0.005
Boundary for River Rch & Prof#=CAMPGROUND CREEK,Reach-1,7
Up Type=0
Dn Type=3
Dn Slope=0.005

--- CAMPGROUND CREEK.g01 (geometry) ---

Geom Title=Existing Conditions
Program Version=4.00

River Reach=CAMPGROUND CREEK,Reach-1
Reach XY= 30
        2870005.       10282716.      2870833.75       10280682.
        2870843.       10279265.      2872165.75       10278905.
      2872885.75       10278044.       2873647.5       10277692.
      2873816.75       10277166.        2875964.       10277995.
        2876603.       10277685.      2876842.25       10276609.
       2877251.5       10276800.      2878660.75       10276519.
       2878487.5       10275593.        2878986.       10275153.
      2880057.75       10272280.        2881339.       10271475.
      2882101.75       10270313.      2883232.75       10269403.
       2884298.5       10269715.       2885673.5       10269162.
      2886111.75       10269510.        2886839.       10269453.
      2887782.75       10270375.       2888776.5       10269822.
        2891121.       10269465.        2893484.       10268572.
       2893846.5       10268133.      2895109.25       10263001.
      2897411.25       10260542.      2899242.25       10259136.

Type RM Length L Ch R = 1 ,47500   ,500,500,500
BEGIN DESCRIPTION:
CAMPGROUND CREEK 95.0
END DESCRIPTION:
XS GIS Cut Line= 3
      2870455.68     10282753.11      2870190.59     10282345.89
      2869705.68     10282303.11
#Sta/Elev= 30
  4514.1 1327.56  4542.8 1326.17  4557.9 1323.35  4563.9 1323.03    4573  1321.2
    4579 1320.96  4609.3 1316.32  4672.5 1310.07  4716.9 1307.12  4729.9 1304.61
  4752.7 1302.94  4775.3 1300.01  4853.7  1294.6  4868.8 1292.38    4905 1289.38
  4926.1 1286.39  4962.4    1284  4989.4 1281.32  4989.6 1280.82  4993.1 1280.82
  4993.4 1281.32    5025 1282.37  5044.5 1283.89  5089.4 1285.48  5095.3 1287.01
  5125.4 1288.24  5175.6 1291.72  5306.1 1302.32  5317.2 1303.72  5486.8 1317.61
#Mann= 5 ,-1 , 0
  4514.1     .12       0  4989.4     .07       0  4993.4     .12       0
  5044.5     .05       0  5317.2     .12       0
Bank Sta=4989.4,4993.4
XS Rating Curve= 0 ,0
Exp/Cntr=0.3,0.1

Type RM Length L Ch R = 1 ,47000   ,292,292,292
BEGIN DESCRIPTION:
CAMPGROUND CREEK 94.0
END DESCRIPTION:
XS GIS Cut Line= 3
      2870655.68     10282003.11      2870384.56     10281886.33
      2869905.68     10281553.11
#Sta/Elev= 30
  4704.8 1297.95  4766.3 1288.35  4771.8 1288.29  4799.7 1284.45  4818.8 1282.97
  4824.6 1281.36  4842.4 1279.22  4865.9 1277.38  4933.4 1274.41    4977 1271.16
  5005.6  1271.1  5013.6 1270.92  5013.9 1270.42  5017.6 1270.92  5045.3 1272.63
  5102.1 1273.28  5217.9 1278.28    5281 1283.65  5303.2 1284.57  5346.4 1289.13
  5382.2 1291.55  5397.1 1293.91    5418 1294.83  5438.9 1297.07  5461.6 1298.31
  5468.6 1299.49  5489.6 1300.34  5534.1 1305.01  5540.2 1304.77  5583.4 1308.28
#Mann= 5 ,-1 , 0
  4704.8     .12       0  4799.7     .05       0  5005.6     .12       0
  5013.6     .05       0  5017.6     .12       0
Bank Sta=5013.6,5017.6
XS Rating Curve= 0 ,0
Exp/Cntr=0.3,0.1

Type RM Length L Ch R = 1 ,46708   ,238,238,238
BEGIN DESCRIPTION:
Mapping XS 03b06da4
END DESCRIPTION:
XS GIS Cut Line= 3
      2870813.08     10281767.43      2870465.88     10281602.52
       2870023.2     10281454.96
#Sta/Elev= 30
  4654.2 1295.45  4677.5 1292.39  4694.6 1291.62  4700.2 1290.23  4739.9 1286.39
  4773.9 1281.98  4784.2 1281.53  4796.6 1278.89  4870.3 1272.83  4894.9 1270.61
  4927.4 1269.46  4939.2 1268.19  5027.4 1265.51  5027.6 1265.01  5031.4 1265.51
  5059.1 1266.11  5148.4 1269.15  5174.8 1271.63    5180 1271.43  5196.9 1273.62
  5260.1 1278.53  5323.4 1284.76  5369.8 1287.77  5396.1 1291.11  5401.4 1290.45
    5433 1293.42  5459.4 1297.25  5464.6  1296.4  5481.5 1298.75  5505.2  1300.2
#Mann= 5 ,-1 , 0
  4654.2     .12       0  4870.3     .05       0  5027.4     .05       0
  5031.4     .05       0  5059.1     .12       0
Bank Sta=5027.4,5031.4
XS Rating Curve= 0 ,0
Exp/Cntr=0.3,0.1

Type RM Length L Ch R = 1 ,46470   ,150,150,150
BEGIN DESCRIPTION:
Mapping XS 001f3ed8
END DESCRIPTION:
XS GIS Cut Line= 3
      2871085.37     10281682.73       2870685.9     10281421.01
      2870116.52     10281274.08
#Sta/Elev= 30
  4404.8 1300.58  4426.9 1298.89  4432.9 1296.95  4463.1 1295.61  4469.1  1293.6
  4484.2 1293.01  4505.3 1289.42  4520.4 1289.25  4526.3 1287.53  4598.7 1282.24
  4628.9 1281.83  4634.9 1279.66  4643.5 1279.93  4758.5 1269.14  4800.7 1266.38
  4954.9 1262.07  4994.2 1256.52  4994.4 1256.02  4998.2 1256.52  5037.5 1260.16
  5094.2 1263.08  5140.8 1267.73  5256.9 1272.02    5275 1274.76  5297.5 1274.77
  5326.7  1277.4    5333 1279.08  5338.2 1278.12  5404.1 1282.91  5470.4 1288.33
#Mann= 4 ,-1 , 0
  4404.8     .12       0  4994.2     .07       0  4998.2     .12       0
  5404.1     .05       0
Bank Sta=4994.2,4998.2
XS Rating Curve= 0 ,0
Exp/Cntr=0.3,0.1

Type RM Length L Ch R = 1 ,46320   ,160,160,160
BEGIN DESCRIPTION:
Mapping XS 451ef735
END DESCRIPTION:
XS GIS Cut Line= 3
      2871195.09     10281524.41      2870639.49     10281255.29
      2870119.64     10281125.33
#Sta/Elev= 30
  4366.5 1276.24  4443.6 1274.28  4449.5 1275.73    4455 1274.05  4500.2 1272.67
  4562.4 1272.31  4658.3 1267.85  4675.3 1268.51  4703.4 1265.84    4743 1264.62
  4748.6 1262.97  4861.5 1260.53  4906.7 1257.26  4912.2 1255.48  4929.2 1255.37
  4934.8 1253.54  4957.4 1251.06  5011.5 1248.51  5011.8 1248.01  5015.5 1248.51
  5054.7 1252.73  5070.2 1256.42  5090.8 1258.98  5219.7 1263.34  5402.5 1273.83
  5420.7  1275.8    5467 1277.17  5472.2 1278.99  5508.3 1280.17  5519.7 1282.06
#Mann= 4 ,-1 , 0
  4366.5     .12       0  5011.5     .07       0  5015.5     .12       0
  5402.5     .05       0
Bank Sta=5011.5,5015.5
XS Rating Curve= 0 ,0
Exp/Cntr=0.3,0.1

Type RM Length L Ch R = 1 ,46160   ,356,356,356
BEGIN DESCRIPTION:
Mapping XS d74afccc
END DESCRIPTION:
XS GIS Cut Line= 4
      2871233.71     10281447.89      2871017.54     10281222.25
      2870244.24     10280947.52      2870043.56      10280973.6
#Sta/Elev= 30
  4341.2 1265.21  4449.2 1260.94  4505.8 1256.71  4555.5 1251.08  4562.4 1252.02
  4576.3 1248.42  4583.5 1248.97  4604.9 1244.86  4647.3 1241.19  4699.7 1240.71
  4725.2 1242.98  4730.5 1241.25  4756.1 1241.21  4843.3 1244.32  4899.7 1243.54
  4997.6  1233.3  5046.3 1230.13  5046.6 1229.63  5050.3 1230.13  5115.7 1234.09
  5141.2 1241.68  5186.3 1247.65  5259.4 1250.82  5295.5  1249.9  5382.8 1260.85
  5473.5 1264.47  5483.4 1266.63  5543.5 1266.96  5583.8 1271.68  5676.7 1277.07
#Mann= 3 ,-1 , 0
  4341.2     .12       0  5046.3     .07       0  5050.3     .12       0
Bank Sta=5046.3,5050.3
XS Rating Curve= 0 ,0
Exp/Cntr=0.3,0.1

Type RM Length L Ch R = 1 ,45804   ,472,472,472
BEGIN DESCRIPTION:
Mapping XS 9a15eb46
END DESCRIPTION:
XS GIS Cut Line= 4
      2871399.99     10281157.07      2870912.65      10280804.1
      2870305.57     10280604.95      2869995.26     10280745.25
#Sta/Elev= 30
  4284.5 1223.63  4312.6 1223.98  4318.7 1222.76  4333.4  1223.8  4404.6 1220.48
  4469.5 1220.16  4490.4 1218.42  4639.2 1216.22  4639.5 1215.72  4643.2 1216.22
  4762.6 1217.45    4792 1219.31    4857 1220.21  4951.7 1218.83  5002.9 1216.27
  5034.7 1216.29  5098.4 1216.89  5193.3 1220.44  5437.3  1218.3  5531.7 1218.26
    5547 1219.78    5601 1220.31  5606.5 1222.09  5612.8 1221.05  5652.7 1222.44
  5750.6 1229.13  5773.7 1229.32    5820 1233.14  5854.3 1237.89  5865.7  1237.7
#Mann= 6 ,-1 , 0
  4284.5     .05       0  4639.2     .07       0  4643.2     .05       0
  4951.7     .12       0  5193.3     .05       0  5437.3     .12       0
Bank Sta=4639.2,4643.2
XS Rating Curve= 0 ,0
Exp/Cntr=0.3,0.1

Type RM Length L Ch R = 1 ,45332   ,338,338,338
BEGIN DESCRIPTION:
Mapping XS 4493eaf0
END DESCRIPTION:
XS GIS Cut Line= 4
      2871444.52     10280916.53      2870874.16     10280309.83
      2870580.29     10280337.38      2870033.93     10280213.42
#Sta/Elev= 30
  4063.5 1207.25  4114.6 1207.28  4121.9 1206.05  4150.2 1205.53    4157 1206.27
  4171.2 1204.66  4376.3 1205.23  4418.8 1203.44    4454 1206.01  4510.7 1207.61
  4595.6 1207.06  4652.3 1204.89  4673.3 1206.04  4680.6 1205.45  4687.5 1206.82
  4694.8 1205.22  4701.6 1206.54  4726.8 1205.98  4864.7 1203.15    4965 1202.56
  5003.1 1200.72  5003.4 1200.22  5007.1 1200.72  5015.2 1202.42  5045.3 1202.35
  5065.4 1204.19  5105.6 1205.05  5415.3 1205.08  5606.2 1207.35  5751.6  1210.6
#Mann= 5 ,-1 , 0
  4063.5     .05       0  4726.8     .12       0  4864.7     .05       0
  5003.1     .03       0  5007.1     .05       0
Bank Sta=5003.1,5007.1
XS Rating Curve= 0 ,0
Exp/Cntr=0.3,0.1

Type RM Length L Ch R = 1 ,44994   ,438,438,438
BEGIN DESCRIPTION:
Mapping XS 06e7337f
END DESCRIPTION:
XS GIS Cut Line= 4
      2871220.49     10280429.01       2870851.2     10279988.42
      2870561.93     10279988.42      2870149.73     10280034.22
#Sta/Elev= 30
  4293.1 1198.93  4371.6 1199.45    4464 1198.99    4542 1199.77  4556.3 1198.92
  4562.9 1199.33  4599.3 1198.86  4620.1 1199.31  4634.4 1198.23  4648.7 1197.89
  4669.5 1198.02  4712.5 1196.91  4741.1 1197.28  4747.6 1196.72  4780.1 1196.32
  4801.3 1196.04  4941.5 1194.62  4941.8 1194.12  4945.3 1194.12  4945.5 1194.62
  5013.5 1195.86  5043.5 1195.15  5204.3 1195.78  5314.5  1196.6  5374.8 1197.63
  5384.9 1198.27    5405 1197.98  5445.3 1199.18  5495.6 1199.14    5572 1201.92
#Mann= 6 ,-1 , 0
  4293.1     .05       0  4780.1     .12       0  4801.3     .05       0
  4941.5     .05       0  4945.5     .05       0  5204.3     .12       0
Bank Sta=4941.5,4945.5
XS Rating Curve= 0 ,0
Exp/Cntr=0.3,0.1

Type RM Length L Ch R = 1 ,44556   ,536,536,536
BEGIN DESCRIPTION:
Mapping XS a238067c
END DESCRIPTION:
XS GIS Cut Line= 5
      2871251.27     10280310.49      2871079.99     10279818.63
      2870899.86      10279578.5      2870626.21      10279561.4
      2870304.78     10279423.64
#Sta/Elev= 30
    4097 1196.19  4254.6 1195.79  4632.2 1189.81  4717.6 1189.66  4873.4 1188.18
  4888.4 1188.06    4903 1188.98  4925.7 1187.22  4972.3 1187.81  4988.4 1186.06
  5000.4 1184.61  5000.6 1184.11  5004.1 1184.11  5004.4 1184.61  5022.4 1186.87
  5072.5 1188.21    5086 1187.36  5112.6 1187.82  5204.8 1186.95  5236.3 1187.87
  5246.5 1186.61    5252 1186.74  5299.1 1189.67  5421.2 1193.47  5427.8 1194.47
  5433.3 1193.93  5464.8 1194.35  5480.4 1193.71    5504 1196.68  5541.9 1197.61
#Mann= 5 ,-1 , 0
    4097     .05       0  4873.4     .12       0  4988.4     .05       0
  5000.4     .03       0  5004.4     .05       0
Bank Sta=5000.4,5004.4
XS Rating Curve= 0 ,0
Exp/Cntr=0.3,0.1

Type RM Length L Ch R = 1 ,44020   ,487,487,487
BEGIN DESCRIPTION:
Mapping XS 7b90efab
END DESCRIPTION:
XS GIS Cut Line= 4
        2871383.     10280064.52      2871278.23     10279487.93
      2871099.15      10279336.4      2870897.13     10278918.59
#Sta/Elev= 30
  4025.5 1189.81    4264 1187.91  4317.4 1186.71  4322.4 1187.23  4429.2 1184.65
  4546.1 1183.51  4555.4 1182.81  4585.9 1182.43  4722.9    1182  4751.5 1180.89
  4850.7 1181.48    4872 1180.88    4949 1180.85  4963.6 1180.32    4972 1179.75
  4984.5 1176.26  4992.2 1174.88  4992.4 1174.38  4995.9 1174.38  4996.2 1174.88
  5001.6 1177.48  5007.1 1177.82  5016.4 1180.52  5029.7 1181.19    5083 1182.37
  5105.2 1183.75  5120.1  1183.9  5127.5  1184.7  5216.3 1186.04  5310.2 1186.17
#Mann= 5 ,-1 , 0
  4025.5     .05       0    4949     .12       0  4963.6     .05       0
  4992.2     .05       0  4996.2     .05       0
Bank Sta=4992.2,4996.2
XS Rating Curve= 0 ,0
Exp/Cntr=0.3,0.1

Type RM Length L Ch R = 1 ,43533   ,541,541,541
BEGIN DESCRIPTION:
Mapping XS 290f0867
END DESCRIPTION:
XS GIS Cut Line= 4
      2871576.23     10279735.21      2871530.77      10279230.8
      2871296.59     10278950.71      2871123.56     10278786.78
#Sta/Elev= 30
  4322.3 1181.78  4364.6 1180.68  4497.8 1180.05  4608.7 1178.68  4665.8 1178.69
  4873.5  1176.2  4923.7 1176.48  4958.1 1176.31  4980.2 1174.21  4986.7 1174.21
    4999 1172.66  4999.3 1172.16  5002.8 1172.16    5003 1172.66  5021.2 1174.27
  5036.2  1176.5  5072.6 1179.18  5079.1 1178.77  5122.1 1180.84  5128.6  1180.6
  5207.1 1183.22  5256.4 1183.73  5277.7 1185.27  5284.7 1184.39  5298.9 1184.18
  5305.8 1183.38  5334.1 1183.78  5351.4 1183.14  5362.2  1182.9  5432.2 1182.69
#Mann= 7 ,-1 , 0
  4322.3     .05       0  4923.7     .12       0    4999     .07       0
    5003     .12       0  5021.2     .05       0  5351.4     .12       0
  5362.2     .05       0
Bank Sta=4999,5003
XS Rating Curve= 0 ,0
Exp/Cntr=0.3,0.1

Type RM Length L Ch R = 1 ,42992   ,441,441,441
BEGIN DESCRIPTION:
Mapping XS c77aefb8
END DESCRIPTION:
XS GIS Cut Line= 4
      2871966.98     10279396.12      2871907.28     10279249.16
      2871838.41     10278803.77      2871604.19     10278675.18
#Sta/Elev= 30
  4513.5 1174.83  4531.6 1174.47  4585.1 1174.66  4633.3 1173.65  4657.1 1173.71
  4667.6 1174.21  4719.5 1173.45    4739 1173.79  4769.3 1172.75  4870.5 1172.06
  4913.8 1171.25  4974.9 1169.26  4975.1 1168.76  4978.6 1168.76  4978.9 1169.26
    4982  1169.7  4991.9 1169.32  5012.2 1171.05  5022.3 1171.03  5052.6 1172.64
  5120.6 1174.62  5176.7  1175.1  5236.4 1176.81  5301.8  1176.9  5317.9 1177.54
  5331.3 1176.73  5339.7 1177.16  5345.4 1176.68  5367.2 1176.52    5390 1177.06
#Mann= 3 ,-1 , 0
  4513.5     .05       0  4974.9     .03       0  4978.9     .05       0
Bank Sta=4974.9,4978.9
XS Rating Curve= 0 ,0
Exp/Cntr=0.3,0.1

Type RM Length L Ch R = 1 ,42551   ,456,456,456
BEGIN DESCRIPTION:
Mapping XS 495403d9
END DESCRIPTION:
XS GIS Cut Line= 4
      2872458.28     10279138.97      2872375.63     10278932.34
      2872214.92     10278776.22      2871994.51     10278574.18
#Sta/Elev= 30
  4621.5 1172.74  4649.4 1171.86  4660.1 1171.02  4672.6 1171.19  4696.8 1170.44
  4703.2 1169.81  4757.1 1167.63  4780.3 1168.16  4821.7 1167.38  4899.9 1167.75
  4970.7 1167.43    4992 1166.01    4999 1165.23  5004.1 1164.05  5004.4 1163.55
  5007.9 1163.55  5008.1 1164.05  5013.1 1166.77  5055.6 1166.21  5097.9    1168
  5119.5 1169.58  5147.9 1170.66  5175.6 1172.36  5254.9 1173.89  5282.3 1174.05
  5289.1 1173.35  5303.3 1174.16  5317.5 1172.97    5360 1172.84  5367.1 1173.23
#Mann= 4 ,-1 , 0
  4621.5     .05       0  5004.1     .05       0  5008.1     .05       0
  5254.9     .12       0
Bank Sta=5004.1,5008.1
XS Rating Curve= 0 ,0
Exp/Cntr=0.3,0.1

Type RM Length L Ch R = 1 ,42095   ,480,480,480
BEGIN DESCRIPTION:
Mapping XS d142bcbe
END DESCRIPTION:
XS GIS Cut Line= 3
      2872761.32     10278978.24      2872646.54     10278707.35
      2872366.43     10278413.46
#Sta/Elev= 30
  4538.4 1170.19  4598.3    1170  4639.4 1168.84  4652.6 1169.31  4663.1  1169.1
  4674.3 1168.23  4685.2 1168.09  4706.9 1166.89  4715.9 1167.29  4774.1 1165.06
  4792.3 1164.71  4797.8 1164.96  4832.2 1163.98  4878.8 1163.62  4892.9 1163.98
  4921.2 1163.37  4991.7 1163.14  4996.9 1161.68  4997.2 1161.18  5000.7 1161.18
  5000.9 1161.68    5020 1163.15    5098 1162.48  5126.2 1162.94  5154.6 1163.74
  5161.5 1164.42    5204 1166.32  5222.8 1166.72  5232.3 1166.51  5238.6 1166.95
#Mann= 5 ,-1 , 0
  4538.4     .05       0  4996.9     .05       0  5000.9     .05       0
  5126.2     .12       0  5222.8     .05       0
Bank Sta=4996.9,5000.9
XS Rating Curve= 0 ,0
Exp/Cntr=0.3,0.1

Type RM Length L Ch R = 1 ,41615   ,460,460,460
BEGIN DESCRIPTION:
Mapping XS 8bf73ddb
END DESCRIPTION:
XS GIS Cut Line= 3
      2872926.63     10278789.99      2872761.33     10278326.24
      2872431.16     10278087.79
#Sta/Elev= 30
    4394 1165.01  4454.4  1164.2  4486.2 1165.28  4571.2 1165.52  4706.7 1161.25
  4751.6 1161.38  4768.3 1160.51  4885.3 1159.58  4914.5 1160.12  4964.8 1159.57
  4979.5 1160.22    4992 1157.71  4998.4 1157.26  4998.7 1156.76  5002.2 1156.76
  5002.4 1157.26  5006.6 1158.71  5015.1 1159.56  5021.3 1161.18    5029 1162.13
  5071.6 1163.97  5078.3 1165.01    5101 1164.79    5128 1166.72  5160.7 1167.99
  5172.2 1168.66  5178.3 1169.88  5201.6 1169.41  5222.5 1170.58  5293.6  1170.8
#Mann= 4 ,-1 , 0
    4394     .05       0  4998.4     .05       0  5002.4     .05       0
  5160.7     .12       0
Bank Sta=4998.4,5002.4
XS Rating Curve= 0 ,0
Exp/Cntr=0.3,0.1

Type RM Length L Ch R = 1 ,41155   ,472,472,472
BEGIN DESCRIPTION:
Mapping XS 959782ca
END DESCRIPTION:
XS GIS Cut Line= 4
      2873032.23     10278652.21      2873013.87     10278137.98
      2872784.29     10278023.19      2872560.12      10277858.5
#Sta/Elev= 30
  4337.5 1161.77  4446.7  1161.6  4546.7 1159.65    4898 1157.42    4973  1157.6
  4995.4 1156.57  5008.2 1155.08  5008.5 1154.58  5012.2 1155.08  5017.7 1157.55
    5027 1158.72  5032.6 1160.42  5049.4 1158.32  5054.9 1160.23  5071.7 1158.62
  5077.3 1159.83  5084.8 1159.16  5094.1 1160.67  5099.7 1160.02  5105.2 1162.24
  5115.3 1162.84  5121.5 1162.26  5129.9 1163.51  5165.4 1165.84  5187.3 1166.31
  5251.1    1168  5257.3 1169.14  5280.4 1168.75  5336.7 1170.41  5386.9 1170.75
#Mann= 5 ,-1 , 0
  4337.5     .05       0    4898     .12       0  5008.2     .07       0
  5012.2     .12       0  5187.3     .05       0
Bank Sta=5008.2,5012.2
XS Rating Curve= 0 ,0
Exp/Cntr=0.3,0.1

Type RM Length L Ch R = 1 ,40683   ,577,577,577
BEGIN DESCRIPTION:
Mapping XS 153862b4
END DESCRIPTION:
XS GIS Cut Line= 5
      2873587.86     10278239.02      2873344.47     10278101.25
      2873280.18     10278000.23      2873206.72     10277747.69
      2873105.71     10277458.45
#Sta/Elev= 30
  4515.3 1160.26  4676.2 1154.09  4695.9  1151.5  4696.1    1151  4699.9  1151.5
  4725.3 1153.94  4828.3 1155.11  4863.9 1154.15  4974.2 1154.51    4982 1154.38
    4995 1152.77  5020.7 1152.72  5047.1 1154.83  5054.2 1156.12  5092.9 1158.53
  5109.6 1160.71  5126.5 1164.41  5131.7 1163.12  5151.3 1164.23  5197.2 1163.35
  5228.3 1160.48  5254.1 1161.21  5259.4 1160.64  5285.1 1162.69  5290.4 1161.94
  5298.5 1162.19  5394.4 1165.44    5404 1166.37  5440.4 1165.97  5484.1 1166.69
#Mann= 4 ,-1 , 0
  4515.3     .05       0  4695.9     .05       0  4699.9     .05       0
  5298.5     .12       0
Bank Sta=4695.9,4699.9
XS Rating Curve= 0 ,0
Exp/Cntr=0.3,0.1

Type RM Length L Ch R = 1 ,40106   ,1308,1308,1308
BEGIN DESCRIPTION:
Mapping XS a9b90c1f
END DESCRIPTION:
XS GIS Cut Line= 5
      2873900.07     10278110.48        2873822.     10277701.78
      2873592.42     10277499.74      2873430.35     10277312.74
      2873102.71     10276987.82
#Sta/Elev= 30
    4425 1163.52  4452.9 1163.59  4528.8 1162.01    4575 1160.14  4628.6 1158.97
  4638.9 1158.86  4829.5  1153.7  4936.8 1152.18  4986.1 1150.42  4993.7 1148.73
  5012.6 1146.85  5012.8 1146.35  5016.3 1146.35  5016.6 1146.85  5022.1 1148.73
    5037 1149.25  5057.3 1150.34  5106.6 1149.53  5186.7 1149.92  5276.6 1151.23
  5298.4    1151  5381.8 1154.09  5418.6 1154.53    5454 1156.19  5588.3 1157.97
  5793.4 1165.84  5807.6 1167.44  5814.6 1167.07  5821.7 1167.97  5855.8 1168.05
#Mann= 8 ,-1 , 0
    4425     .05       0  4628.6     .12       0  4638.9     .05       0
  5012.6     .05       0  5016.6     .05       0    5037     .12       0
  5186.7     .05       0  5381.8     .12       0
Bank Sta=5012.6,5016.6
XS Rating Curve= 0 ,0
Exp/Cntr=0.3,0.1

Type RM Length L Ch R = 1 ,38798   ,372,372,372
BEGIN DESCRIPTION:
CAMPGROUND CREEK 77.0
END DESCRIPTION:
XS GIS Cut Line= 3
      2874055.69      10278503.1      2874505.68     10277453.11
       2874644.7     10276896.67
#Sta/Elev= 30
    3869 1170.92  4258.8 1160.19  4663.2 1155.28    4685 1153.57  4924.6 1145.21
  4929.5 1145.32  4989.6 1143.22  5000.3 1140.77  5000.5 1140.27  5004.3 1140.77
  5008.6 1142.26  5028.8 1143.38  5062.9 1142.78  5111.9 1144.84    5117 1143.45
  5128.9  1144.1  5158.3  1143.3  5194.4 1145.12  5240.8 1144.44  5276.9 1146.62
  5318.1 1147.29  5382.4 1151.17  5405.7 1149.21  5441.8 1149.03  5454.6 1147.41
  5475.2 1149.44  5483.1 1151.18  5495.8 1156.29    5537 1160.47  5584.9 1162.44
#Mann= 7 ,-1 , 0
    3869     .05       0  4924.6     .12       0  4929.5     .05       0
  5000.3     .05       0  5004.3     .05       0  5028.8     .12       0
  5128.9     .05       0
Bank Sta=5000.3,5004.3
XS Rating Curve= 0 ,0
Exp/Cntr=0.3,0.1

Type RM Length L Ch R = 1 ,38426   ,426,426,426
BEGIN DESCRIPTION:
Mapping XS b722e28a
END DESCRIPTION:
XS GIS Cut Line= 3
      2874441.55     10277991.43       2874832.2     10277566.06
      2874814.86     10277097.72
#Sta/Elev= 30
  4354.3 1156.34  4377.5  1156.1  4398.5 1154.61  4433.6 1154.62  4447.8 1153.33
  4476.1  1152.3  4511.9 1151.87  4589.6 1149.07  4660.5 1147.79  4717.2 1145.57
  4766.5  1145.2  4787.5 1144.03  4894.2 1142.09  4915.1 1140.62  4964.8  1141.4
  4971.3 1142.16  4994.8 1139.78  5012.8 1139.56  5013.1 1139.06  5016.6 1139.06
  5016.8 1139.56  5034.9 1140.82  5044.9 1140.38  5084.9    1144  5144.9 1147.85
    5225 1150.47    5265 1152.28  5325.1 1153.49  5385.1 1150.81  5400.5 1149.29
#Mann= 4 ,-1 , 0
  4354.3     .05       0  5012.8     .05       0  5016.8     .05       0
    5225     .12       0
Bank Sta=5012.8,5016.8
XS Rating Curve= 0 ,0
Exp/Cntr=0.3,0.1

Type RM Length L Ch R = 1 ,38000   ,500,500,500
BEGIN DESCRIPTION:
CAMPGROUND CREEK 76.0
END DESCRIPTION:
XS GIS Cut Line= 3
      2874355.71     10278203.09      2875189.56     10277572.07
      2875155.69     10277203.12
#Sta/Elev= 30
  3954.3 1159.76    4076 1157.22  4182.1 1153.02    4205 1153.31  4246.6 1151.53
  4396.4 1149.47  4460.9 1147.08  4589.9 1144.85  4718.9 1140.42  4775.1 1136.93
  4789.7 1137.31  4795.9 1135.81  4845.9  1137.6  4889.5 1136.68  4932.4 1133.73
  4968.6 1134.26  4980.6 1133.29  4980.8 1132.79  4984.6 1133.29    5019    1134
  5059.2 1138.45  5100.7 1137.24  5119.5 1140.29  5149.6 1141.42  5189.8 1144.74
  5206.7 1144.97  5219.9 1144.87  5290.2 1152.54  5315.6 1156.31  5370.5 1160.95
#Mann= 4 ,-1 , 0
  3954.3     .05       0  4980.6     .05       0  4984.6     .05       0
  5206.7     .12       0
Bank Sta=4980.6,4984.6
XS Rating Curve= 0 ,0
Exp/Cntr=0.3,0.1

Type RM Length L Ch R = 1 ,37500   ,510,510,510
BEGIN DESCRIPTION:
CAMPGROUND CREEK 75.0
END DESCRIPTION:
XS GIS Cut Line= 3
       2875005.7     10278453.09      2875568.08     10277805.63
      2875505.68     10277453.11
#Sta/Elev= 30
  4142.4 1148.28  4298.6 1144.02  4383.1 1138.54  4433.4 1141.13  4532.2 1133.92
  4574.9 1135.39  4624.3 1132.91  4631.9 1136.12  4652.8 1137.11  4844.4 1139.82
  4900.6 1137.21  4914.9 1135.69  4922.5 1133.08  4929.1 1134.35  4936.7 1131.68
  4978.5 1132.07  4986.1  1129.8  4992.7 1130.05  4996.4 1127.61  4996.6 1127.11
  5000.4 1127.61  5022.9 1131.61  5045.3 1131.79  5063.5  1134.3  5083.8 1134.48
  5114.3 1137.17  5158.6 1142.68    5165 1144.81  5297.1 1148.88    5358 1148.28
#Mann= 3 ,-1 , 0
  4142.4     .05       0  4996.4     .05       0  5000.4     .05       0
Bank Sta=4996.4,5000.4
XS Rating Curve= 0 ,0
Exp/Cntr=0.3,0.1

Type RM Length L Ch R = 1 ,36990   ,288,288,288
BEGIN DESCRIPTION:
Mapping XS 2450957b
END DESCRIPTION:
XS GIS Cut Line= 4
      2875873.33      10278271.2      2875942.79      10278058.5
       2875934.1     10277828.46      2875886.36     10277620.12
#Sta/Elev= 30
  4712.7 1136.74  4768.6 1134.79  4773.8 1135.33  4794.8 1134.42  4805.7 1134.99
  4832.4 1132.56  4837.6 1133.58    4858 1132.83  4864.2 1131.84  4869.5 1132.48
  4889.5 1131.19  4901.4  1129.1  4910.6 1126.22    4928 1128.77  4981.9 1128.65
  4989.5 1125.48  4994.5 1125.88  4999.9 1125.09  5000.1 1124.59  5003.9 1125.09
  5071.9 1127.94  5081.9 1127.09    5092 1127.22  5161.8 1131.49  5184.8 1130.95
  5222.5 1132.08  5227.7 1131.36  5270.6 1133.39  5318.6 1132.83  5380.4 1133.25
#Mann= 3 ,-1 , 0
  4712.7     .05       0  4999.9     .05       0  5003.9     .05       0
#XS Ineff= 2 , 0
       0  4981.9                       0
Permanent Ineff=
       F       F
Bank Sta=4999.9,5003.9
XS Rating Curve= 0 ,0
Exp/Cntr=0.3,0.1

Type RM Length L Ch R = 1 ,36702   ,387,387,387
BEGIN DESCRIPTION:
Mapping XS 7d2b37cc
END DESCRIPTION:
XS GIS Cut Line= 4
      2876025.27     10278336.23      2876172.82     10278010.75
       2876181.5     10277780.72      2876107.72     10277533.35
#Sta/Elev= 30
  4525.8 1138.08  4559.9 1138.49  4565.4 1137.86    4628 1139.33    4672 1138.74
  4732.5 1135.95    4738 1137.13  4755.6 1135.84  4778.7 1135.79  4900.8 1130.82
  4940.8 1128.18  4950.9 1126.84  4960.9 1123.58  4968.9 1122.44  4969.1 1121.94
  4972.9 1122.44  5030.9 1125.09  5040.9 1126.99  5060.9 1128.32  5093.8 1126.94
  5131.7 1127.86  5182.4 1127.69  5204.8 1129.05    5226 1128.11  5246.5 1129.77
  5267.4 1129.13  5325.5 1130.77  5330.7 1129.97  5350.9 1131.87  5371.5 1132.12
#Mann= 3 ,-1 , 0
  4525.8     .05       0  4968.9     .03       0  4972.9     .05       0
Bank Sta=4968.9,4972.9
XS Rating Curve= 0 ,0
Exp/Cntr=0.3,0.1

Type RM Length L Ch R = 1 ,36315   ,152,152,152
BEGIN DESCRIPTION:
Mapping XS fb408f8e
END DESCRIPTION:
XS GIS Cut Line= 4
      2876828.17     10278145.27      2876632.89     10277919.61
      2876311.71     10277559.36      2875912.42     10277212.15
#Sta/Elev= 30
  4527.9 1129.35  4559.2 1128.97  4623.3 1130.51  4701.8 1129.53  4751.1 1131.35
  4826.3 1130.28  4871.6 1131.75  4914.3 1131.29    4921 1132.36  4935.2 1131.77
  4949.4 1128.98  4956.1 1129.47    4992 1121.69  4996.7 1121.54    4997 1121.04
  5000.7 1121.54  5034.7  1125.3  5048.9 1124.09  5076.5 1124.12  5090.7 1125.73
  5147.5 1126.12  5225.3 1129.23  5402.7 1130.53  5416.9 1131.78  5423.6 1130.87
  5459.7 1132.93  5551.8 1135.16  5629.6 1135.02  5750.2 1138.38  5838.1 1142.14
#Mann= 3 ,-1 , 0
  4527.9     .05       0  4996.7     .03       0  5000.7     .05       0
Bank Sta=4996.7,5000.7
XS Rating Curve= 0 ,0
Exp/Cntr=0.3,0.1

Type RM Length L Ch R = 1 ,36163   ,663,663,663
BEGIN DESCRIPTION:
Mapping XS 7e4a8126
END DESCRIPTION:
XS GIS Cut Line= 3
      2876910.68     10278010.76      2876463.62     10277507.28
      2876116.37     10277190.42
#Sta/Elev= 30
  4543.5 1127.98  4637.3 1129.14  4773.6 1127.92  4800.3 1127.44  4830.3 1128.52
  4849.7 1128.85  4878.1 1126.78  4899.8 1123.63  4920.8 1123.11    4935 1124.82
  4955.9 1124.64  4970.1 1122.15  4977.6 1122.88  4984.3 1120.59  4991.8 1122.89
  4996.5 1119.32  4996.8 1118.82  5000.5 1119.32  5041.2 1124.37    5098 1126.17
  5104.7 1127.13  5126.5 1126.88  5133.2 1127.91  5140.7 1126.42  5154.9  1126.4
  5366.8 1129.44  5494.5 1133.52  5501.3 1134.74    5558 1137.06  5686.9 1138.33
#Mann= 5 ,-1 , 0
  4543.5     .05       0  4773.6     .12       0  4830.3     .05       0
  4996.5     .03       0  5000.5     .05       0
Bank Sta=4996.5,5000.5
XS Rating Curve= 0 ,0
Exp/Cntr=0.3,0.1

Type RM Length L Ch R = 1 ,35500   ,500,500,500
BEGIN DESCRIPTION:
CAMPGROUND CREEK 71.0
END DESCRIPTION:
XS GIS Cut Line= 3
       2877805.7     10278053.13       2876676.5      10277068.8
      2876155.66      10276703.1
#Sta/Elev= 30
    3502 1142.55  3601.2 1141.68  3776.4 1135.63  3991.4 1127.46  4380.6  1124.1
  4497.6 1124.71  4707.2 1124.44  4856.2 1122.45  4921.8 1122.74  4940.8 1122.89
    4955 1118.64  4961.7    1120  4973.2 1117.26  4973.6 1116.76  4978.6 1117.26
    5019 1119.44  5033.8 1123.43  5054.7 1122.62  5111.3 1126.25    5120 1128.17
  5227.2 1130.64  5283.9  1134.4  5298.7 1134.13  5313.5 1130.88  5328.3 1131.18
  5334.4 1132.95    5364 1133.25    5506 1140.61    5629  1144.9  5636.4 1143.89
#Mann= 8 ,-1 , 0
    3502     .12       0  3776.4     .05       0  4497.6     .12       0
  4856.2     .05       0  4921.8     .12       0  4973.2     .07       0
  4978.6     .12       0    5506     .05       0
Bank Sta=4973.2,4978.6
XS Rating Curve= 0 ,0
Exp/Cntr=0.3,0.1

Type RM Length L Ch R = 1 ,35000   ,500,500,500
BEGIN DESCRIPTION:
CAMPGROUND CREEK 70.0
END DESCRIPTION:
XS GIS Cut Line= 3
      2877705.69     10277903.13      2876835.41     10276614.47
      2876505.67     10276553.11
#Sta/Elev= 30
    3445 1140.54  3491.5 1138.94  3553.6 1136.28  3611.3 1135.38  3638.4 1133.77
  3878.1 1127.06    3986  1126.4  4150.9 1127.82  4374.2 1124.41  4525.5 1120.24
    4537 1120.89  4753.6 1119.56  4957.1 1121.11  4965.4  1120.3  4978.1  1117.2
  4995.1 1115.78  4995.5 1115.28  5000.5 1115.78  5009.9 1116.17    5030 1122.72
    5035 1126.56  5070.9 1131.12  5087.8 1129.05  5092.9 1130.25  5101.4 1129.69
    5132 1131.12  5145.6  1133.5    5193 1135.65  5303.9 1137.43  5335.4 1136.57
#Mann= 6 ,-1 , 0
    3445     .12       0  3491.5     .05       0    4537     .12       0
  4753.6     .05       0  4995.1     .03       0  5000.5     .05       0
Bank Sta=4995.1,5000.5
XS Rating Curve= 0 ,0
Exp/Cntr=0.3,0.1

Type RM Length L Ch R = 1 ,34500   ,500,500,500
BEGIN DESCRIPTION:
CAMPGROUND CREEK 69.0
END DESCRIPTION:
XS GIS Cut Line= 3
       2877605.7     10277753.14      2877247.73     10276799.41
      2877005.68     10275803.09
#Sta/Elev= 30
  3981.3 1134.49  4332.8  1125.7  4718.3 1122.08  4820.3 1121.72  4825.7 1122.81
  4845.2 1121.42  4921.3 1120.99  4974.7 1119.76  4985.4 1117.29  4991.2 1114.24
  5003.7 1113.85  5004.1 1113.35  5009.3 1113.85  5047.6 1117.47  5072.8 1118.55
  5088.8 1117.53  5140.3  1118.8    5274 1118.81  5323.4 1124.92  5365.1 1126.94
  5453.8 1126.98  5531.3 1125.48  5542.5 1124.96  5562.2  1120.4  5579.1 1121.92
  5629.3 1122.82  5850.7 1129.65  5932.7 1133.34  5973.8 1133.06  6025.3 1134.56
#Mann= 5 ,-1 , 0
  3981.3     .05       0  5003.7     .05       0  5009.3     .05       0
  5629.3     .12       0  5850.7     .05       0
Bank Sta=5003.7,5009.3
XS Rating Curve= 0 ,0
Exp/Cntr=0.3,0.1

Type RM Length L Ch R = 1 ,34000   ,500,500,500
BEGIN DESCRIPTION:
CAMPGROUND CREEK 68.0
END DESCRIPTION:
XS GIS Cut Line= 3
      2877705.68     10277703.13      2877677.09     10276738.35
      2877255.68     10275753.09
#Sta/Elev= 30
  4034.8 1135.53    4415 1125.16  4540.6  1123.3    4555 1123.79  4585.1 1122.61
  4635.1  1122.6  4865.2 1118.64  4955.2 1118.46    5000 1116.51  5005.7 1112.75
  5010.9 1111.78  5011.4 1111.28  5016.5 1111.78  5049.2 1115.05  5060.1 1114.65
  5089.9 1116.94    5119 1116.54  5136.2 1117.43  5234.1 1116.26  5347.6 1123.23
  5376.6 1123.18  5423.8 1121.45  5462.5 1118.24    5471 1119.35  5494.6 1118.85
  5628.8 1120.48  5728.6 1122.69  5799.4 1125.94  5957.3 1129.91  6071.6 1133.95
#Mann= 3 ,-1 , 0
  4034.8     .05       0  5010.9     .03       0  5016.5     .05       0
Bank Sta=5010.9,5016.5
XS Rating Curve= 0 ,0
Exp/Cntr=0.3,0.1

Type RM Length L Ch R = 1 ,33500   ,500,500,500
BEGIN DESCRIPTION:
CAMPGROUND CREEK 67.0
END DESCRIPTION:
XS GIS Cut Line= 3
      2878755.71     10277153.13       2878102.6     10276482.09
       2877555.7     10275653.14
#Sta/Elev= 30
  4063.6 1133.58  4473.8 1121.88  4530.4 1120.69  4629.4 1121.16  4721.2  1115.4
  4770.8 1113.61  4848.5 1113.37  4961.7  1115.1  4980.2 1109.85  4980.7 1109.35
  4985.8 1109.85  5025.2 1110.76  5034.3 1112.56  5040.3 1111.91  5046.7 1114.06
  5055.3 1114.72  5142.5 1114.16  5184.8 1116.22  5258.3 1114.86  5286.3 1114.29
  5335.3 1116.25  5358.2 1114.92    5432 1117.04  5629.8  1122.8  5772.1  1126.1
    5820 1128.41    5826  1127.6  5938.8 1130.95  5956.2 1131.36  5993.1 1132.53
#Mann= 9 ,-1 , 0
  4063.6     .05       0  4980.2     .03       0  4985.8     .05       0
  5258.3     .12       0    5432     .05       0  5629.8     .12       0
  5772.1     .05       0  5938.8     .12       0  5956.2     .05       0
Bank Sta=4980.2,4985.8
XS Rating Curve= 0 ,0
Exp/Cntr=0.3,0.1

Type RM Length L Ch R = 1 ,33000   ,500,500,500
BEGIN DESCRIPTION:
CAMPGROUND CREEK 66.0
END DESCRIPTION:
XS GIS Cut Line= 3
      2878805.68     10276953.11      2878554.88     10276549.25
      2877555.69     10275553.12
#Sta/Elev= 30
  4524.6 1131.58  4642.1 1128.42  4742.5 1122.08  4830.7 1123.59  4910.2 1118.12
  4924.8 1113.79  4931.4 1113.67  4952.7 1119.35  4989.3 1114.97  4994.8 1111.02
    5000 1111.02  5000.9 1107.96  5001.4 1107.46  5006.7 1107.96  5109.8 1108.79
  5116.9 1110.72    5124 1109.75    5131 1112.52  5138.1 1110.09  5145.2 1112.66
  5152.3 1111.28  5159.3 1113.42  5298.1 1113.16    5322 1111.72  5378.5 1116.32
  5512.9 1113.17  5781.6 1115.16    5939 1119.26  6024.6 1121.38  6410.9 1134.45
#Mann= 7 ,-1 , 0
  4524.6     .05       0  5000.9     .03       0  5006.7     .05       0
  5298.1     .12       0  5781.6     .05       0    5939     .12       0
  6024.6     .05       0
Bank Sta=5000.9,5006.7
XS Rating Curve= 0 ,0
Exp/Cntr=0.3,0.1

Type RM Length L Ch R = 1 ,32500   ,500,500,500
BEGIN DESCRIPTION:
CAMPGROUND CREEK 65.0
END DESCRIPTION:
XS GIS Cut Line= 3
      2879305.64      10276353.1      2878644.69     10276146.81
      2877655.68     10275603.11
#Sta/Elev= 30
  4307.6 1126.91    4339 1126.67  4421.3  1123.3  4691.7 1115.27  4915.2 1116.49
  4956.9 1110.88  4967.5 1110.36  4988.5 1106.33  5019.8 1106.14  5020.3 1105.64
  5025.6 1106.14  5044.5 1106.87  5090.2  1106.5  5098.5 1108.94  5104.2 1108.21
    5113 1110.18  5136.8  1110.5  5201.7 1110.14    5251  1111.9    5338 1112.31
  5457.5 1111.45    5555 1114.62  5582.5 1113.91  5598.6 1115.55  5604.3 1114.32
  5658.3 1115.06  5761.5  1118.5  5797.7 1121.31  5957.6 1124.88  6128.6 1131.67
#Mann= 5 ,-1 , 0
  4307.6     .05       0  5019.8     .03       0  5025.6     .05       0
  5136.8     .12       0    5338     .05       0
Bank Sta=5019.8,5025.6
XS Rating Curve= 0 ,0
Exp/Cntr=0.3,0.1

Type RM Length L Ch R = 1 ,32000   ,487,487,487
BEGIN DESCRIPTION:
CAMPGROUND CREEK 64.0
END DESCRIPTION:
XS GIS Cut Line= 3
      2879405.67      10276353.1      2878480.11      10275683.8
      2877755.65      10275453.1
#Sta/Elev= 30
  3857.8 1129.98  4008.9 1125.76  4110.5 1123.36  4294.4 1120.61  4537.3 1113.47
  4545.8 1112.57  4602.3 1112.72  4732.2 1109.49  4931.4  1108.9  4954.2 1105.71
  4993.1  1103.9  4993.6  1103.4  4998.9  1103.9  4999.6 1105.87  5019.6 1107.49
  5025.6 1108.81  5046.5 1108.59  5057.1 1106.63  5067.6 1106.17  5077.9 1107.03
    5084 1108.49  5089.3 1108.03  5099.1    1109  5163.2 1109.38  5384.7 1115.06
  5481.1 1118.88  5550.8 1124.13  5621.5 1127.17  5634.3 1128.56  5760.3  1131.5
#Mann= 9 ,-1 , 0
  3857.8     .05       0  4008.9     .12       0  4110.5     .05       0
  4993.1     .03       0  4998.9     .05       0  5077.9     .12       0
  5163.2     .05       0  5384.7     .12       0  5621.5     .05       0
Bank Sta=4993.1,4998.9
XS Rating Curve= 0 ,0
Exp/Cntr=0.3,0.1

Type RM Length L Ch R = 1 ,31513   ,513,513,513
BEGIN DESCRIPTION:
Mapping XS 4e589776
END DESCRIPTION:
XS GIS Cut Line= 4
      2879280.45     10275684.36      2878794.35     10275315.44
      2878490.53     10275167.87      2878191.02     10275102.76
#Sta/Elev= 30
  4281.6 1115.69  4442.7  1111.6  4457.2 1112.02  4507.1 1110.46  4571.6 1110.07
  4677.7 1106.31  4756.7 1104.93  4827.5 1106.03  4930.4 1106.05  4935.9 1105.15
  4975.5  1105.3  5000.5  1101.5    5001    1101  5006.8  1101.5  5012.6 1102.94
  5020.6 1103.44  5034.9 1102.55  5048.7 1104.05  5110.9 1105.43  5116.4 1104.94
  5123.8 1105.65  5178.6 1106.17  5184.1 1105.02  5206.7 1106.46  5223.7 1105.95
    5273 1108.74  5278.1 1110.45  5285.7 1109.63    5296 1109.79  5536.1 1116.14
#Mann= 3 ,-1 , 0
  4281.6     .05       0  5000.5     .03       0  5006.8     .05       0
Bank Sta=5000.5,5006.8
XS Rating Curve= 0 ,0
Exp/Cntr=0.3,0.1

Type RM Length L Ch R = 1 ,31000   ,372,372,372
BEGIN DESCRIPTION:
CAMPGROUND CREEK 62.0
END DESCRIPTION:
XS GIS Cut Line= 3
      2879405.66     10275103.11      2879003.65     10274990.09
      2878505.69     10274803.11
#Sta/Elev= 30
  4582.4 1119.71  4599.4 1119.84  4638.7 1115.03  4655.1 1116.81  4717.4  1112.4
    4746 1115.19  4751.2 1112.35  4769.4 1114.47  4790.5 1112.63  4819.3 1116.34
  4824.5 1113.42  4858.6 1115.97  4883.6 1111.91  4897.8 1105.79  4956.3 1104.21
  4996.3 1097.96  5026.1 1097.17  5026.6 1096.67  5032.5 1097.17  5059.5 1100.88
  5150.3  1103.2  5190.1 1109.15  5211.5 1105.53  5243.5 1109.23  5376.2 1111.14
  5401.1 1117.28  5406.5 1113.09  5478.5 1118.18  5499.9 1117.09  5531.9 1120.78
#Mann= 3 ,-1 , 0
  4582.4     .05       0  5026.1     .03       0  5032.5     .05       0
Bank Sta=5026.1,5032.5
XS Rating Curve= 0 ,0
Exp/Cntr=0.3,0.1

Type RM Length L Ch R = 1 ,30628   ,446,446,446
BEGIN DESCRIPTION:
Mapping XS a99cd727
END DESCRIPTION:
XS GIS Cut Line= 4
      2879640.74     10274768.58      2879380.29     10274694.78
      2878894.17     10274607.98      2878542.59     10274577.59
#Sta/Elev= 30
  4406.4 1109.94  4453.2 1109.92  4519.5  1108.8  4567.6 1107.55    4578 1107.79
  4626.5 1105.97  4676.9 1104.97  4828.9 1102.79  4864.6  1101.4  4895.1 1098.88
  4915.4 1098.33  4941.7 1096.72    4956 1097.09  4966.2 1096.75  4983.3 1095.11
  4983.8 1094.61  4989.2 1094.61  4989.7 1095.11  5006.8 1096.07    5017 1097.88
  5037.3 1099.72  5054.5 1099.15  5077.9 1100.04  5113.4 1099.82  5209.5 1102.46
  5269.8 1103.28  5285.1 1104.02  5309.9 1104.05  5470.5 1107.95  5523.8 1109.71
#Mann= 3 ,-1 , 0
  4406.4     .05       0  4983.3     .03       0  4989.7     .05       0
Bank Sta=4983.3,4989.7
XS Rating Curve= 0 ,0
Exp/Cntr=0.3,0.1

Type RM Length L Ch R = 1 ,30182   ,682,682,682
BEGIN DESCRIPTION:
Mapping XS beb15476
END DESCRIPTION:
XS GIS Cut Line= 4
      2879931.46      10274495.1      2879605.98     10274304.16
      2879080.81     10274213.01      2878633.71     10274191.31
#Sta/Elev= 30
  4248.7 1103.81  4416.3 1102.31    4555 1100.44  4576.5 1099.61  4591.6 1100.06
  4603.7 1099.28    4781  1097.1  4798.9 1096.28  4849.6 1095.48  4920.7 1095.49
  4949.9 1094.31  5009.6 1093.15  5011.5 1092.71    5012 1092.21  5017.4 1092.21
  5017.9 1092.71  5042.5 1094.44  5062.8 1094.12  5074.4 1094.52  5083.1 1092.93
  5093.2 1092.84  5113.5 1095.04    5144 1094.42  5184.2 1095.97  5414.5 1100.05
  5454.6 1101.81  5484.6 1104.38  5494.6 1103.92  5524.6 1104.55  5606.7  1104.1
#Mann= 3 ,-1 , 0
  4248.7     .05       0  5011.5     .03       0  5017.9     .05       0
Bank Sta=5011.5,5017.9
XS Rating Curve= 0 ,0
Exp/Cntr=0.3,0.1

Type RM Length L Ch R = 1 ,29500   ,500,500,500
BEGIN DESCRIPTION:
CAMPGROUND CREEK 59.0
END DESCRIPTION:
XS GIS Cut Line= 3
      2880255.71     10274253.13      2879452.15     10273615.36
       2879034.8     10273379.87
#Sta/Elev= 30
  3974.1  1106.2  4002.2 1107.44  4066.2 1106.25  4074.3 1107.04  4095.1 1105.79
  4216.7 1104.17  4237.7 1102.73  4394.7 1100.01  4444.4 1098.36  4550.1 1096.62
    4579 1097.43  4678.3 1094.31  4714.6 1092.29  4906.1 1089.27  4920.2 1089.17
  4928.2 1090.15  4949.1 1088.89  4960.2 1086.66  4960.7 1086.16  4966.8 1086.66
  4977.9 1088.48  5007.4 1088.16  5019.7 1086.95  5029.9 1088.32  5057.3 1088.14
  5073.2  1090.1  5078.9 1089.68  5132.4 1092.64  5256.6 1095.67  5479.2 1092.78
#Mann= 3 ,-1 , 0
  3974.1     .05       0  4960.2     .05       0  4966.8     .05       0
Bank Sta=4960.2,4966.8
XS Rating Curve= 0 ,0
Exp/Cntr=0.3,0.1

Type RM Length L Ch R = 1 ,29000   ,500,500,500
BEGIN DESCRIPTION:
CAMPGROUND CREEK 58.0
END DESCRIPTION:
XS GIS Cut Line= 4
      2880255.71     10273753.13      2879732.38     10273266.82
      2879486.68     10273201.91      2879009.95     10272791.93
#Sta/Elev= 30
  4285.6 1103.76  4589.8 1098.74  4681.6 1095.11    4710 1095.04  4717.3 1094.02
  4802.3 1091.79  4823.3 1089.55  4886.8 1087.07  4979.2 1085.77  4993.4 1083.67
  5024.3 1082.57  5024.8 1082.07  5030.9 1082.57  5048.3 1085.39  5073.7 1086.02
  5089.7  1087.4  5172.4 1087.09  5275.3 1088.67  5445.3 1085.66  5473.9 1085.98
  5494.7 1084.51    5509 1087.02  5750.4 1094.67  5764.6 1096.17  5778.9 1095.84
  5835.8 1098.45  5842.6 1099.08  5849.2 1101.11  5863.4 1102.38  5882.9 1102.09
#Mann= 3 ,-1 , 0
  4285.6     .05       0  5024.3     .03       0  5030.9     .05       0
Bank Sta=5024.3,5030.9
XS Rating Curve= 0 ,0
Exp/Cntr=0.3,0.1

Type RM Length L Ch R = 1 ,28500   ,370,370,370
BEGIN DESCRIPTION:
CAMPGROUND CREEK 57.0
END DESCRIPTION:
XS GIS Cut Line= 3
      2880305.68      10273653.1       2879968.9     10272849.62
      2879250.69     10272548.73
#Sta/Elev= 30
  4128.8 1101.55  4373.6  1096.9  4486.6 1092.98  4540.8 1093.26  4692.6 1089.77
  4863.4 1082.76  4887.1 1082.94  4892.6 1080.68  4898.6  1080.1  4921.8 1081.18
  4936.8 1079.19  4937.3 1078.69  4943.5 1079.19  4945.5 1081.88  4993.1  1079.5
  5006.4 1079.65  5024.8 1082.51  5083.2 1080.39  5130.7 1083.11  5242.1 1083.38
  5337.3 1086.83  5372.1 1089.68  5437.2 1089.74  5549.2 1092.35  5567.3 1091.63
    5679 1093.17  5719.1 1094.71  5755.7  1094.7  5773.3  1095.3  5778.7 1096.46
#Mann= 3 ,-1 , 0
  4128.8     .05       0  4936.8     .03       0  4943.5     .05       0
#XS Ineff= 2 , 0
       0                 5024.74       0
Permanent Ineff=
       F       F
Bank Sta=4936.8,4943.5
XS Rating Curve= 0 ,0
Exp/Cntr=0.3,0.1

Type RM Length L Ch R = 1 ,28130   ,630,630,630
BEGIN DESCRIPTION:
Mapping XS e1dea201
END DESCRIPTION:
XS GIS Cut Line= 4
      2880465.34      10272889.2       2880200.6     10272546.34
      2879840.35     10272407.45      2879245.76     10272259.89
#Sta/Elev= 30
  4423.3 1091.48  4463.1 1088.89  4620.5  1084.8  4712.2 1083.43  4726.7 1084.08
  4747.5 1082.53    4820 1080.87  4847.9 1079.42  4878.6 1080.02  4893.9 1078.91
    4926 1080.15  4963.2 1079.67  4975.9 1077.31  4976.4 1076.81  4983.4 1077.31
  5017.7 1077.43  5077.7 1079.27    5097 1077.75  5126.9    1080  5132.3 1079.54
  5186.9 1081.22  5277.2 1085.12  5350.4 1086.55  5453.4 1086.24  5463.7 1086.88
  5489.2 1085.84  5546.2 1086.76  5587.4 1085.73  5742.6 1090.68  5855.2  1092.4
#Mann= 3 ,-1 , 0
  4423.3     .05       0  4975.9     .03       0  4983.4     .05       0
Bank Sta=4975.9,4983.4
XS Rating Curve= 0 ,0
Exp/Cntr=0.3,0.1

Type RM Length L Ch R = 1 ,27500   ,500,500,500
BEGIN DESCRIPTION:
CAMPGROUND CREEK 55.0
END DESCRIPTION:
XS GIS Cut Line= 3
       2880605.7     10272553.14      2880406.01     10272068.14
      2879905.71     10271703.13
#Sta/Elev= 30
  4475.5 1091.37  4484.8  1091.6  4538.1 1086.83  4591.4 1085.25  4644.7 1081.64
  4703.4 1079.82  4713.4 1080.31  4735.1 1078.12  4789.1 1076.08  4821.6 1075.95
  4843.2 1074.28  4864.8 1074.98  4881.9  1073.7  4897.3 1074.01  4940.6  1072.3
  4988.5 1072.36  4999.5 1070.29    5000 1069.79  5007.2 1070.29  5047.3 1073.23
  5074.7 1073.98  5124.6 1072.92  5147.8 1073.56  5189.5 1077.43  5233.5 1079.72
  5260.5 1082.86    5347 1087.25  5433.7 1088.98  5540.9 1089.21  5619.3 1092.71
#Mann= 3 ,-1 , 0
  4475.5     .05       0  4999.5     .05       0  5007.2     .05       0
Bank Sta=4999.5,5007.2
XS Rating Curve= 0 ,0
Exp/Cntr=0.3,0.1

Type RM Length L Ch R = 1 ,27000   ,500,500,500
BEGIN DESCRIPTION:
CAMPGROUND CREEK 54.0
END DESCRIPTION:
XS GIS Cut Line= 3
      2880805.68     10272553.14      2880779.25     10271750.87
      2880405.67      10271403.1
#Sta/Elev= 30
  4197.3 1089.73  4227.3 1089.68  4297.4 1084.57  4417.4  1079.7  4597.5 1075.47
  4707.6 1074.65  4857.7 1069.84  4941.2 1069.02  4977.7 1067.44  4987.8 1066.41
  4992.5 1064.53    4993 1064.03  5000.3 1064.53  5007.9 1065.31  5015.2 1064.54
    5022  1066.7  5036.2  1067.6  5042.7 1067.06  5060.8 1068.14  5092.9 1067.58
  5142.2 1069.41  5149.6 1070.61  5163.7 1070.48  5241.4 1074.39  5248.8  1076.3
  5262.9 1075.33  5342.3 1078.64  5411.4 1081.48  5439.8 1081.68  5510.4 1085.64
#Mann= 7 ,-1 , 0
  4197.3     .05       0  4941.2     .12       0  4992.5     .07       0
  5000.3     .12       0  5042.7     .05       0  5060.8     .12       0
  5342.3     .05       0
Bank Sta=4992.5,5000.3
XS Rating Curve= 0 ,0
Exp/Cntr=0.3,0.1

Type RM Length L Ch R = 1 ,26500   ,500,500,500
BEGIN DESCRIPTION:
CAMPGROUND CREEK 53.0
END DESCRIPTION:
XS GIS Cut Line= 3
      2881555.68     10272053.11      2881223.11     10271537.09
      2880705.68     10271053.11
#Sta/Elev= 30
  4386.1 1082.98  4393.7 1081.12    4430 1078.74  4523.7 1075.44  4647.8  1073.3
  4762.7 1067.34  4820.1  1066.8  4835.3  1064.7  4898.7 1063.02    4929 1061.19
    4931 1060.12  4931.5 1059.62  4938.9 1060.12  4950.2 1061.11  5008.2 1060.26
  5043.4 1062.87  5085.9 1063.47  5142.6 1063.64  5163.6 1062.55  5199.2 1065.12
  5255.9 1066.79  5361.9 1068.37  5425.4 1070.64  5453.7 1072.92  5461.1 1074.74
  5467.9 1073.85  5510.4 1074.83  5637.9  1081.5  5687.2 1082.29  5708.5 1084.16
#Mann= 3 ,-1 , 0
  4386.1     .05       0    4931     .03       0  4938.9     .05       0
Bank Sta=4931,4938.9
XS Rating Curve= 0 ,0
Exp/Cntr=0.3,0.1

Type RM Length L Ch R = 1 ,26000   ,500,500,500
BEGIN DESCRIPTION:
CAMPGROUND CREEK 52.0
END DESCRIPTION:
XS GIS Cut Line= 3
      2881605.67     10271403.08      2881524.17     10271161.57
      2881155.65     10270953.09
#Sta/Elev= 30
  4745.1 1070.94  4755.5 1071.34  4760.8 1068.76  4766.2 1069.39  4829.5 1063.93
  4855.2 1062.72  4881.4 1059.37  4886.7 1060.22  4903.4 1057.11  4924.5 1056.65
  4949.6 1054.36  4975.8 1054.12  4981.1 1052.82    5000 1052.89  5001.5 1050.22
    5002 1049.72  5009.5 1050.22  5021.2 1050.39  5032.9 1052.82  5055.7  1053.8
  5064.7 1056.08  5070.4 1055.11  5086.3 1061.59  5092.1  1059.7    5108 1063.07
  5136.1 1064.84  5188.8 1064.09  5210.5 1065.77  5226.4 1065.05  5423.4 1072.12
#Mann= 3 ,-1 , 0
  4745.1     .05       0  5001.5     .05       0  5009.5     .05       0
Bank Sta=5001.5,5009.5
XS Rating Curve= 0 ,0
Exp/Cntr=0.3,0.1

Type RM Length L Ch R = 1 ,25500   ,500,500,500
BEGIN DESCRIPTION:
CAMPGROUND CREEK 51.0
END DESCRIPTION:
XS GIS Cut Line= 3
      2881955.69     10271403.13      2881748.64     10270733.82
      2881555.68      10270253.1
#Sta/Elev= 30
  4299.4 1069.89  4341.3 1070.56  4362.2 1068.31    4381 1068.62  4418.8 1066.65
    4446 1068.12  4456.7 1066.51  4498.3 1066.41  4540.2 1065.04  4554.5 1065.49
  4690.3  1059.5  4948.4 1050.65  4969.3 1048.77  5003.1 1048.37  5015.1  1046.4
  5015.6  1045.9  5023.2  1046.4  5043.3 1050.59  5119.3 1055.02  5258.5    1061
  5263.9 1062.08  5288.1 1061.49  5293.5 1062.25  5312.3 1061.84  5317.7 1063.08
  5334.8 1062.43  5385.8 1063.04  5454.8 1064.88  5515.1 1070.86    5518 1070.88
#Mann= 5 ,-1 , 0
  4299.4     .05       0  5015.1     .03       0  5023.2     .05       0
  5385.8     .12       0  5515.1     .05       0
Bank Sta=5015.1,5023.2
XS Rating Curve= 0 ,0
Exp/Cntr=0.3,0.1

Type RM Length L Ch R = 1 ,25000   ,500,500,500
BEGIN DESCRIPTION:
CAMPGROUND CREEK 50.0
END DESCRIPTION:
XS GIS Cut Line= 3
      2882422.79     10270740.76      2882092.62     10270442.27
      2881905.71     10270253.14
#Sta/Elev= 30
  4554.9 1062.94  4742.1 1053.14  4756.3 1051.93  4770.5 1049.13  4798.9 1048.56
  4806.4 1049.38  4813.1 1048.55  4827.3 1049.56  4834.1 1050.99  4898.3 1050.82
    4905  1050.1  4926.7 1050.74  4946.6 1045.88  4957.8 1045.23  4958.3 1044.73
  4965.9 1045.23    5000 1046.01  5004.3 1047.23  5011.4 1046.73  5018.4  1048.5
  5032.6 1047.27  5060.9 1047.25    5068 1045.75    5075 1047.52  5103.3 1049.97
  5117.4 1054.43  5138.7 1057.88  5195.3 1062.24  5216.4 1062.39  5265.9 1065.84
#Mann= 4 ,-1 , 0
  4554.9     .05       0  4946.6     .12       0  4957.8     .07       0
  4965.9     .12       0
Bank Sta=4957.8,4965.9
XS Rating Curve= 0 ,0
Exp/Cntr=0.3,0.1

Type RM Length L Ch R = 1 ,24500   ,500,500,500
BEGIN DESCRIPTION:
CAMPGROUND CREEK 49.0
END DESCRIPTION:
XS GIS Cut Line= 3
      2882605.68     10270703.11      2882419.39     10270195.09
      2881905.69     10270003.11
#Sta/Elev= 30
  4458.9 1065.06  4490.8 1064.79  4554.8  1062.8  4732.7 1054.55  4746.5 1053.48
  4809.5 1051.63  4831.7 1050.58  4878.1 1050.05  4935.5 1049.52  4959.5 1047.23
  4984.4 1042.54    4987 1042.27  4987.5 1041.77  4994.8 1041.77  4995.3 1042.27
  4996.5 1043.21  5004.6 1043.05  5014.6 1043.82  5021.3  1043.3    5036  1046.6
  5105.5 1050.86  5135.8 1052.11  5153.4 1051.92  5281.9 1056.89  5331.9 1060.16
  5356.2 1060.42  5441.9 1064.79  5472.7 1066.99    5503 1067.19  5548.4 1069.89
#Mann= 8 ,-1 , 0
  4458.9     .05       0  4809.5     .12       0  4878.1     .05       0
  4984.4     .12       0    4987     .07       0  4995.3     .12       0
  5021.3     .05       0  5441.9     .12       0
Bank Sta=4987,4995.3
XS Rating Curve= 0 ,0
Exp/Cntr=0.3,0.1
