--- BENNETT CREEK.prj (project) ---

Proj Title=BENNETT CREEK Base Level Engineering
Current Plan=p01
Default Exp/Contr=0.3,0.1
English Units
Geom File=g01
Flow File=f01
Plan File=p01
Y Axis Title=Elevation
X Axis Title(PF)=Main Channel Distance
X Axis Title(XS)=Station
BEGIN DESCRIPTION:
BENNETT CREEK
END DESCRIPTION:
DSS Export Rating Curves= 0
DSS Export Rating Curve Sorted= 0
DSS Export Volume Flow Curves= 0
DXF OffsetX= 0
DXF OffsetY= 0
DXF ScaleX= 1
DXF ScaleY= 10

--- BENNETT CREEK.p01 (plan) ---

Plan Title=Multiple Run
Short Identifier=Multiple
Geom File=g01
Flow File=f01
Subcritical Flow
K Sum by GR= 0
Std Step Tol= 0.01
Critical Tol= 0.01
Num of Std Step Trials= 20
Max Error Tol= 0.3
Flow Tol Ratio= 0.001
Split Flow NTrial= 30
Split Flow Tol= 0.02
Split Flow Ratio= 0.02
Log Output Level= 0
Friction Slope Method= 1
Unsteady Friction Slope Method= 2
Unsteady Bridges Friction Slope Method= 1
Parabolic Critical Depth
Global Vel Dist=  1 , 1 , 1
Global Log Level= 0
CheckData=True
Encroach Param= -1, 0, 0, 0
BEGIN DESCRIPTION:
Multiple Run
END DESCRIPTION:

--- BENNETT CREEK.f01 (steady flow) ---

Flow Title=Multiple
Program Version=4.10
Number of Profiles= 7
Profile Names=10-year,25-year,50-year,1pct_min,100-year,1pct_plu,500-year
River Rch & RM=BENNETT CREEK,Reach-1         ,50000
     754    1267    1317     890    1730    3363    2292
River Rch & RM=BENNETT CREEK,Reach-1         ,40500
     924    1574    1753    1185    2334    4599    3107
River Rch & RM=BENNETT CREEK,Reach-1         ,38000
    1395    2435    2971    1999    4040    8164    5392
River Rch & RM=BENNETT CREEK,Reach-1         ,32219
    1559    2744    3378    2249    4617    9479    6169
River Rch & RM=BENNETT CREEK,Reach-1         ,29000
    1697    2999    3808    2548    5230   10735    6994
River Rch & RM=BENNETT CREEK,Reach-1         ,28000
    1900    3392    4331    2847    5985   12579    8028
River Rch & RM=BENNETT CREEK,Reach-1         ,23500
    2056    3687    4761    3127    6599   13928    8848
River Rch & RM=BENNETT CREEK,Reach-1         ,21500
    2442    4448    5675    3620    7919   17324   10642
River Rch & RM=BENNETT CREEK,Reach-1         ,12500
    2664    4887    6429    4073    9039   20058   12211
River Rch & RM=BENNETT CREEK,Reach-1         ,7500
    3149    5881    8318    5321   11842   26358   15949
River Rch & RM=BENNETT CREEK,Reach-1         ,2500
    3235    6059    8538    5433   12164   27236   16375
Boundary for River Rch & Prof#=BENNETT CREEK,Reach-1         , 1
Up Type= 0
Dn Type= 3
Dn Slope=0.0005
Boundary for River Rch & Prof#=BENNETT CREEK,Reach-1         , 2
Up Type= 0
Dn Type= 3
Dn Slope=0.0005
Boundary for River Rch & Prof#=BENNETT CREEK,Reach-1         , 3
Up Type= 0
Dn Type= 3
Dn Slope=0.0005
Boundary for River Rch & Prof#=BENNETT CREEK,Reach-1         , 4
Up Type= 0
Dn Type= 3
Dn Slope=0.0005
Boundary for River Rch & Prof#=BENNETT CREEK,Reach-1         , 5
Up Type= 0
Dn Type= 3
Dn Slope=0.0005
Boundary for River Rch & Prof#=BENNETT CREEK,Reach-1         , 6
Up Type= 0
Dn Type= 3
Dn Slope=0.0005
Boundary for River Rch & Prof#=BENNETT CREEK,Reach-1         , 7
Up Type= 0
Dn Type= 3
Dn Slope=0.0005
DSS Import GetInterval= 0
DSS Import GetPeak= 0
DSS Import FillOption= 0

--- BENNETT CREEK.g01 (geometry) ---

Geom Title=Existing Conditions

River Reach=BENNETT CREEK,Reach-1
Reach XY= 30
      2780808.75     10189577.00      2780128.00     10191627.00
      2779477.25     10191807.00      2779285.75     10193070.00
      2778621.00     10193226.00      2777469.75     10194765.00
      2777885.75     10196084.00      2777421.00     10199007.00
      2776517.25     10200534.00      2776700.25     10201355.00
      2775071.00     10203028.00      2776474.25     10205488.00
      2775963.75     10207780.00      2773436.75     10209368.00
      2774466.00     10210697.00      2774570.00     10212897.00
      2774103.50     10212740.00      2773932.50     10211695.00
      2773474.25     10211797.00      2773072.25     10214101.00
      2772286.75     10214168.00      2772849.25     10215263.00
      2771272.00     10215472.00      2771628.25     10217205.00
      2770549.25     10217953.00      2771240.00     10221025.00
      2770546.25     10221858.00      2771125.25     10222761.00
      2770313.00     10223379.00      2770187.25     10224186.00

Type RM Length L Ch R = 1,50000,500,500,500
BEGIN DESCRIPTION:
BENNETT CREEK 100.0
END DESCRIPTION:
XS GIS Cut Line= 3
      2779805.71     10189053.12      2780816.78     10189612.09
      2781755.68     10190553.11
#Sta/Elev= 30
  3844.7 1383.50  4198.9 1371.19  4574.3 1368.83  4587.4 1367.63  4815.9 1365.26
  4851.5 1364.31  4867.6 1362.29  4873.3 1363.32  4941.6 1360.25  5019.0 1360.04
  5019.3 1359.54  5023.4 1360.04  5042.4 1360.32  5063.6 1368.82  5070.7 1369.78
  5091.9 1363.38  5115.9 1362.57  5147.5 1362.85  5229.3 1364.00  5403.0 1367.74
  5657.6 1368.60  5799.0 1371.66  5890.9 1375.54  5933.3 1375.53  6131.3 1384.29
  6216.2 1391.48  6230.3 1391.66  6237.4 1389.59  6265.7 1394.65  6329.3 1399.33
#Mann=7,-1,0
  3844.7    0.05       0  4867.6    0.12       0  5019.0    0.07       0
  5023.4    0.12       0  5115.9    0.05       0  5147.5    0.12       0
  5229.3    0.05       0
Bank Sta=5019,5023.4
Exp/Cntr=0.3,0.1

Type RM Length L Ch R = 1,49500,500,500,500
BEGIN DESCRIPTION:
BENNETT CREEK 99.0
END DESCRIPTION:
XS GIS Cut Line= 3
      2779705.67     10189103.10      2780691.02     10190078.25
      2781655.70     10191053.13
#Sta/Elev= 30
  3613.7 1383.26  3748.1 1379.90  3903.6 1373.10  3988.5 1370.83  4002.6 1371.70
  4009.7 1370.10  4200.6 1368.42  4398.6 1373.14  4660.2 1366.13  4674.4 1364.65
  4897.8 1362.18  4947.2 1361.14  4978.4 1361.23  5011.5 1357.96  5011.8 1357.46
  5016.1 1357.96  5056.2 1361.36  5445.1 1366.54  5593.7 1370.34  5636.1 1372.91
  5643.1 1371.92  5791.7 1378.29  5996.7 1392.27  6017.9 1391.63  6025.0 1393.89
  6056.0 1396.94  6109.8 1403.57  6279.5 1419.69  6300.8 1423.10  6371.5 1429.19
#Mann=6,-1,0
  3613.7    0.05       0  4897.8    0.12       0  4947.2    0.05       0
  5011.5    0.05       0  5016.1    0.05       0  6056.0    0.12       0
Bank Sta=5011.5,5016.1
Exp/Cntr=0.3,0.1

Type RM Length L Ch R = 1,49000,500,500,500
BEGIN DESCRIPTION:
BENNETT CREEK 98.0
END DESCRIPTION:
XS GIS Cut Line= 3
      2778555.67     10189253.10      2780550.62     10190507.21
      2781505.66     10191303.10
#Sta/Elev= 30
  2643.6 1402.55  2868.0 1390.05  3151.5 1379.45  3347.3 1375.44  3645.3 1374.91
  3876.2 1368.75  3950.6 1367.00  3996.4 1366.11  4072.9 1365.66  4108.3 1363.29
  4143.7 1365.66  4381.2 1364.66  4619.6 1361.34  4921.3 1359.32  4985.6 1359.16
  4997.6 1357.17  4998.0 1356.67  5002.3 1357.17  5163.5 1363.29  5434.2 1367.36
  5675.0 1377.10  5810.4 1388.16  5831.2 1387.39  5839.0 1390.16  5938.3 1402.06
  6051.2 1414.26  6100.7 1422.22  6193.1 1430.58  6230.5 1436.59  6243.2 1438.95
#Mann=11,-1,0
  2643.6    0.05       0  3876.2    0.12       0  3950.6    0.05       0
  3996.4    0.12       0  4381.2    0.05       0  4619.6    0.12       0
  4921.3    0.05       0  4997.6    0.05       0  5002.3    0.05       0
  5938.3    0.12       0  6230.5    0.05       0
Bank Sta=4997.6,5002.3
Exp/Cntr=0.3,0.1

Type RM Length L Ch R = 1,48500,500,500,500
BEGIN DESCRIPTION:
BENNETT CREEK 97.0
END DESCRIPTION:
XS GIS Cut Line= 3
      2779155.65     10190053.08      2780132.43     10190746.53
      2781105.72     10191703.14
#Sta/Elev= 30
  3802.1 1380.52  3986.0 1371.95  4081.8 1369.13  4204.4 1366.52  4412.3 1365.33
  4525.7 1362.78  4555.0 1363.59  4783.8 1358.90  4820.0 1356.52  4854.9 1356.98
  4918.0 1355.73  4918.3 1355.23  4922.7 1355.73  4953.4 1357.23  4985.5 1356.11
  5035.2 1358.25  5211.1 1358.45  5452.9 1360.62  5714.1 1365.96  5890.8 1372.18
  5975.7 1375.98  6011.1 1379.04  6039.4 1377.48  6110.1 1382.80  6131.3 1382.01
  6195.0 1386.27  6237.4 1392.24  6286.9 1396.74  6332.7 1406.00  6364.7 1411.02
#Mann=10,-1,0
  3802.1    0.05       0  3986.0    0.12       0  4081.8    0.05       0
  4854.9    0.12       0  4918.0    0.05       0  4922.7    0.12       0
  4953.4    0.05       0  5211.1    0.12       0  5452.9    0.05       0
  6332.7    0.12       0
Bank Sta=4918,4922.7
Exp/Cntr=0.3,0.1

Type RM Length L Ch R = 1,48000,500,500,500
BEGIN DESCRIPTION:
BENNETT CREEK 96.0
END DESCRIPTION:
XS GIS Cut Line= 3
      2779405.72     10190753.14      2779888.02     10191094.88
      2780855.68     10191603.11
#Sta/Elev= 30
  4408.9 1375.85  4445.6 1374.86  4458.0 1375.67  4466.7 1374.43  4492.1 1374.17
  4536.0 1372.38  4595.3 1369.22  4757.9 1362.16  4811.2 1359.90  4974.9 1356.31
  5008.1 1353.19  5008.5 1352.69  5013.1 1353.19  5019.9 1354.77  5032.7 1353.81
  5071.1 1356.13  5087.5 1355.85  5093.2 1354.65  5131.6 1356.68  5159.3 1355.55
  5279.7 1355.16  5641.2 1361.70  5759.7 1365.19  5908.4 1372.62  5936.1 1372.91
  6002.6 1376.11  6018.7 1378.30  6025.2 1376.86  6040.7 1376.52  6093.0 1381.00
#Mann=7,-1,0
  4408.9    0.05       0  4492.1    0.12       0  4536.0    0.05       0
  4595.3    0.12       0  4757.9    0.05       0  5008.1    0.05       0
  5013.1    0.05       0
Bank Sta=5008.1,5013.1
Exp/Cntr=0.3,0.1

Type RM Length L Ch R = 1,47500,500,500,500
BEGIN DESCRIPTION:
BENNETT CREEK 95.0
END DESCRIPTION:
XS GIS Cut Line= 3
      2779155.73     10190953.13      2780162.25     10191493.71
      2780555.68     10191903.11
#Sta/Elev= 30
  3857.5 1381.28  4166.8 1366.73  4183.0 1367.01  4300.1 1361.91  4314.5 1362.55
  4402.3 1358.65  4595.3 1356.00  4653.9 1356.44  4839.8 1353.49  4981.2 1353.91
  5006.6 1350.81  5007.0 1350.31  5011.7 1350.81  5016.1 1353.45  5030.2 1355.69
  5044.4 1356.57  5122.3 1357.68  5249.4 1361.71  5263.6 1363.83  5277.7 1369.65
  5284.9 1369.95  5299.1 1369.24  5306.0 1366.51  5334.3 1361.64  5405.1 1361.07
  5426.4 1362.72  5461.7 1368.94  5539.6 1372.14  5553.8 1373.74  5567.8 1373.54
#Mann=3,-1,0
  3857.5    0.05       0  5006.6    0.05       0  5011.7    0.05       0
Bank Sta=5006.6,5011.7
Exp/Cntr=0.3,0.1

Type RM Length L Ch R = 1,47000,500,500,500
BEGIN DESCRIPTION:
BENNETT CREEK 94.0
END DESCRIPTION:
XS GIS Cut Line= 3
      2779105.71     10191053.14      2779804.48     10191745.53
      2780755.66     10192703.09
#Sta/Elev= 30
  4016.3 1381.30  4171.8 1375.94  4419.3 1364.04  4751.6 1353.62  4893.1 1351.21
  4963.8 1351.73  4982.5 1348.57  4982.9 1348.07  4987.6 1348.57  5006.2 1353.32
  5034.5 1352.00  5076.9 1353.87  5260.8 1356.18  5282.0 1357.99  5303.2 1356.67
  5359.8 1357.17  5550.7 1361.20  5692.1 1367.66  5713.3 1367.19  5876.0 1375.71
  5911.3 1374.64  5925.5 1377.00  6024.5 1384.91  6045.7 1384.89  6066.9 1389.39
  6165.9 1403.62  6223.3 1416.73  6270.7 1424.02  6314.4 1433.38  6349.7 1437.41
#Mann=5,-1,0
  4016.3    0.05       0  4982.5    0.05       0  4987.6    0.05       0
  6223.3    0.12       0  6270.7    0.05       0
Bank Sta=4982.5,4987.6
Exp/Cntr=0.3,0.1

Type RM Length L Ch R = 1,46500,500,500,500
BEGIN DESCRIPTION:
BENNETT CREEK 93.0
END DESCRIPTION:
XS GIS Cut Line= 3
      2779055.67     10191103.08      2779477.07     10191954.39
      2780405.72     10192753.14
#Sta/Elev= 30
  4050.1 1382.55  4064.1 1382.07  4081.0 1378.88  4148.3 1375.82  4467.9 1366.37
  4641.5 1360.49  4675.3 1358.07  4781.9 1356.85  4864.7 1357.84  4894.0 1356.47
  4922.0 1352.51  4938.9 1352.80  4966.9 1349.15  4983.7 1349.16  4993.9 1346.62
  4994.3 1346.12  4999.0 1346.62  5019.5 1349.47  5068.9 1350.77  5275.2 1353.90
  5431.0 1354.26  5494.6 1356.82  5565.3 1356.08  5777.7 1362.04  6019.1 1370.99
  6097.0 1376.16  6125.6 1375.47  6139.8 1377.74  6217.7 1382.77  6224.9 1384.52
#Mann=3,-1,0
  4050.1    0.05       0  4993.9    0.05       0  4999.0    0.05       0
Bank Sta=4993.9,4999
Exp/Cntr=0.3,0.1

Type RM Length L Ch R = 1,46000,500,500,500
BEGIN DESCRIPTION:
BENNETT CREEK 92.0
END DESCRIPTION:
XS GIS Cut Line= 3
      2778305.66     10191853.10      2779330.67     10192420.98
      2780255.67     10193353.10
#Sta/Elev= 30
  3828.2 1373.35  3954.0 1368.30  3998.8 1367.99  4011.1 1366.52  4239.8 1359.88
  4297.6 1356.81  4351.4 1356.47  4410.9 1354.00  4497.9 1352.57  4880.0 1350.50
  4982.9 1347.78  4991.3 1345.35  5009.5 1343.94  5009.9 1343.44  5014.7 1343.94
  5019.2 1345.68  5054.6 1347.61  5167.7 1347.75  5224.3 1349.04  5280.8 1351.96
  5344.5 1352.37  5478.8 1356.99  5648.5 1358.77  5761.7 1361.60  5797.0 1363.74
  5818.3 1363.34  6157.7 1376.46  6228.4 1380.09  6235.4 1381.44  6313.2 1384.39
#Mann=3,-1,0
  3828.2    0.05       0  5009.5   0.035       0  5014.7    0.05       0
Bank Sta=5009.5,5014.7
Exp/Cntr=0.3,0.1

Type RM Length L Ch R = 1,45500,500,500,500
BEGIN DESCRIPTION:
BENNETT CREEK 91.0
END DESCRIPTION:
XS GIS Cut Line= 3
      2778355.71     10192803.11      2779347.61     10192906.75
      2779605.71     10193003.12
#Sta/Elev= 30
  4002.7 1364.65  4083.1 1361.75  4103.2 1360.41  4123.3 1357.85  4147.7 1356.38
  4153.5 1355.52  4294.3 1348.64  4314.4 1348.35  4364.6 1346.17  4425.0 1346.44
  4465.2 1345.79  4565.7 1347.21  4676.3 1346.91  4728.0 1348.02  4736.6 1347.48
  4797.0 1347.57  4816.3 1349.34  4837.2 1346.94  4897.5 1343.48  4914.7 1341.73
  4993.9 1341.51  4994.3 1341.01  4998.8 1341.01  4999.2 1341.51  5033.9 1341.66
  5058.9 1348.98  5089.2 1353.86  5222.1 1361.80  5254.1 1362.19  5275.5 1361.60
#Mann=3,-1,0
  4002.7    0.05       0  4993.9    0.05       0  4999.2    0.05       0
Bank Sta=4993.9,4999.2
Exp/Cntr=0.3,0.1

Type RM Length L Ch R = 1,45000,500,500,500
BEGIN DESCRIPTION:
BENNETT CREEK 90.0
END DESCRIPTION:
XS GIS Cut Line= 3
      2778305.72     10192903.12      2778985.32     10193169.37
      2779955.72     10194103.15
#Sta/Elev= 30
  4270.1 1366.29  4463.4 1352.01  4592.3 1345.96  4719.1 1343.10  4941.5 1342.65
  4946.9 1341.50  4966.0 1341.46  4993.1 1339.78  4993.5 1339.28  4998.4 1339.78
  5031.1 1342.60  5158.5 1346.64  5427.3 1352.78  5604.0 1355.36  5660.6 1357.79
  5681.7 1357.07  5780.8 1359.69  5802.1 1361.42  5865.7 1362.37  5929.5 1365.59
  5964.7 1365.61  6007.2 1368.60  6028.3 1367.91  6035.5 1369.17  6141.5 1372.64
  6198.1 1376.73  6205.3 1378.15  6240.5 1378.68  6286.9 1384.42  6346.7 1392.99
#Mann=4,-1,0
  4270.1    0.05       0  4993.1    0.03       0  4998.4    0.05       0
  6286.9    0.12       0
Bank Sta=4993.1,4998.4
Exp/Cntr=0.3,0.1

Type RM Length L Ch R = 1,44500,500,500,500
BEGIN DESCRIPTION:
BENNETT CREEK 89.0
END DESCRIPTION:
XS GIS Cut Line= 3
      2778255.72     10193003.14      2778593.99     10193348.88
      2779555.71     10194303.13
#Sta/Elev= 30
  4516.3 1363.16  4636.5 1357.21  4685.9 1352.09  4799.1 1345.37  4855.6 1343.05
  4933.5 1342.65  4961.8 1341.31  4990.1 1338.19  4994.3 1335.51  4994.7 1335.01
  4999.8 1335.51  5004.7 1335.65  5011.3 1338.71  5018.3 1338.40  5025.4 1340.05
  5188.0 1340.33  5237.5 1341.69  5485.0 1343.54  5866.9 1351.49  6008.3 1355.24
  6050.7 1357.39  6079.0 1357.41  6114.4 1358.87  6135.6 1360.85  6163.8 1360.82
  6262.8 1364.99  6269.9 1366.22  6312.4 1367.61  6319.4 1366.91  6354.8 1368.80
#Mann=3,-1,0
  4516.3    0.05       0  4994.3    0.03       0  4999.8    0.05       0
Bank Sta=4994.3,4999.8
Exp/Cntr=0.3,0.1

Type RM Length L Ch R = 1,44000,500,500,500
BEGIN DESCRIPTION:
BENNETT CREEK 88.0
END DESCRIPTION:
XS GIS Cut Line= 3
      2778055.70     10193453.12      2778560.74     10193781.49
      2779505.65     10194753.08
#Sta/Elev= 30
  4397.6 1359.11  4519.8 1352.19  4564.6 1346.83  4643.7 1341.29  4737.2 1338.12
  4933.6 1338.56  4994.0 1334.24  4994.5 1333.74  4999.7 1334.24  5011.7 1334.45
  5018.7 1337.06  5047.0 1336.81  5110.8 1341.45  5372.4 1350.57  5457.3 1352.58
  5627.0 1349.16  5718.9 1350.16  5810.9 1352.62  5895.6 1357.79  5987.6 1359.36
  6008.8 1361.67  6030.1 1360.62  6121.9 1365.04  6129.1 1363.91  6192.7 1368.89
  6249.3 1371.19  6277.5 1375.70  6313.0 1378.81  6330.6 1383.76  6355.3 1386.98
#Mann=4,-1,0
  4397.6    0.05       0  4994.0    0.05       0  4999.7    0.05       0
  6330.6    0.12       0
Bank Sta=4994,4999.7
Exp/Cntr=0.3,0.1

Type RM Length L Ch R = 1,43500,500,500,500
BEGIN DESCRIPTION:
BENNETT CREEK 87.0
END DESCRIPTION:
XS GIS Cut Line= 3
      2777955.68     10193703.10      2778134.92     10193905.16
      2779105.65     10194553.09
#Sta/Elev= 30
  4729.9 1355.70  4751.2 1354.63  4772.1 1351.66  4836.5 1345.64  4843.2 1343.55
  4921.0 1338.63  4928.5 1336.24  4989.2 1331.88  4989.7 1331.38  4994.9 1331.88
  5002.7 1332.08  5006.1 1333.77  5012.9 1334.80  5049.0 1335.92  5252.4 1338.80
  5360.6 1339.54  5396.6 1341.14  5423.7 1340.87  5546.8 1344.18  5561.9 1345.20
  5691.0 1349.25  5742.1 1349.53  5829.2 1348.08  5835.2 1349.71  5907.3 1349.48
  5958.4 1350.70  5979.4 1350.51  5994.4 1351.40  6015.4 1351.01  6167.1 1355.24
#Mann=3,-1,0
  4729.9    0.05       0  4989.2    0.05       0  4994.9    0.05       0
Bank Sta=4989.2,4994.9
Exp/Cntr=0.3,0.1

Type RM Length L Ch R = 1,43000,500,500,500
BEGIN DESCRIPTION:
BENNETT CREEK 86.0
END DESCRIPTION:
XS GIS Cut Line= 3
      2777605.70     10193903.14      2777785.84     10194234.10
      2779705.71     10194953.12
#Sta/Elev= 30
  4623.2 1355.88  4748.4 1350.94  4828.1 1343.07  4941.8 1336.16  4993.7 1328.63
  4994.2 1328.13  4999.4 1328.63  5021.2 1331.58  5043.9 1332.51  5202.7 1333.68
  5551.5 1341.06  5758.1 1350.16  5863.1 1350.67  5953.9 1347.36  6046.3 1346.19
  6345.3 1353.53  6547.0 1361.55  6590.9 1365.24  6612.9 1364.17  6622.9 1368.52
  6740.4 1382.32  6772.4 1388.36  6778.5 1392.10  6811.8 1396.03  6857.9 1404.15
  6894.2 1406.44  6919.2 1411.01  6979.7 1417.26  7019.3 1419.62  7050.1 1422.94
#Mann=5,-1,0
  4623.2    0.05       0  4993.7    0.05       0  4999.4    0.05       0
  6811.8    0.12       0  7019.3    0.05       0
Bank Sta=4993.7,4999.4
Exp/Cntr=0.3,0.1

Type RM Length L Ch R = 1,42500,500,500,500
BEGIN DESCRIPTION:
BENNETT CREEK 85.0
END DESCRIPTION:
XS GIS Cut Line= 3
      2777305.65     10194603.11      2777661.26     10194658.51
      2778481.57     10194799.29
#Sta/Elev= 30
  4640.1 1348.24  4680.6 1345.76  4781.8 1336.82  4791.9 1335.63  4799.8 1333.83
  4812.2 1332.72  4862.6 1330.44  4872.9 1328.52  4893.1 1329.28  4964.0 1329.70
  4990.5 1327.18  4991.0 1326.68  4995.8 1326.68  4996.3 1327.18  4998.4 1328.07
  5014.6 1328.65  5045.1 1332.72  5053.5 1333.16  5233.5 1339.13  5288.4 1339.26
  5339.3 1337.59  5413.5 1337.32  5430.6 1337.74  5440.8 1338.87  5461.1 1337.30
  5533.5 1338.78  5633.6 1342.87  5703.3 1345.03  5745.2 1345.35  5832.3 1343.92
#Mann=3,-1,0
  4640.1    0.05       0  4990.5    0.05       0  4996.3    0.05       0
Bank Sta=4990.5,4996.3
Exp/Cntr=0.3,0.1

Type RM Length L Ch R = 1,42000,500,500,500
BEGIN DESCRIPTION:
BENNETT CREEK 84.0
END DESCRIPTION:
XS GIS Cut Line= 3
      2777050.09     10194960.88      2777419.00     10195025.36
      2778888.67     10195341.10
#Sta/Elev= 30
  4625.5 1335.94  4781.0 1338.95  4840.5 1339.16  4894.9 1337.91  4959.5 1334.16
  4976.3 1331.18  4995.8 1324.05  5003.9 1322.75  5004.4 1322.25  5009.7 1322.75
  5012.5 1324.47  5047.7 1328.40  5098.9 1329.47  5150.0 1326.51  5170.5 1326.67
  5211.4 1329.63  5392.2 1335.31  5548.9 1331.23  5584.6 1331.03  5628.8 1332.87
  5702.4 1333.83  5821.2 1332.30  5835.3 1330.45  5870.6 1332.93  6183.1 1345.01
  6316.0 1351.67  6428.6 1355.38  6449.0 1357.53  6479.7 1357.03  6503.2 1358.45
#Mann=3,-1,0
  4625.5    0.05       0  5003.9    0.05       0  5009.7    0.05       0
Bank Sta=5003.9,5009.7
Exp/Cntr=0.3,0.1

Type RM Length L Ch R = 1,41500,500,500,500
BEGIN DESCRIPTION:
BENNETT CREEK 83.0
END DESCRIPTION:
XS GIS Cut Line= 3
      2776605.66     10195803.12      2777629.37     10195451.25
      2778555.73     10195653.12
#Sta/Elev= 30
  3917.5 1351.22  4058.1 1346.97  4115.3 1343.62  4490.2 1329.97  4541.4 1327.58
  4573.1 1324.21  4584.0 1324.25  4594.3 1327.05  4604.6 1328.05  4698.4 1333.90
  4859.9 1330.39  4917.1 1326.48  4953.8 1322.11  4979.6 1321.35  4992.5 1318.53
  4993.0 1318.03  4998.3 1318.53  5032.4 1325.58  5076.1 1327.04  5141.1 1326.67
  5241.9 1326.78  5344.2 1324.92  5518.2 1334.24  5551.4 1334.58  5600.5 1338.43
  5794.5 1346.28  5845.7 1350.27  5874.4 1349.36  5886.6 1353.17  5948.1 1355.98
#Mann=5,-1,0
  3917.5    0.05       0  4992.5    0.03       0  4998.3    0.05       0
  5032.4    0.12       0  5141.1    0.05       0
Bank Sta=4992.5,4998.3
Exp/Cntr=0.3,0.1

Type RM Length L Ch R = 1,41000,500,500,500
BEGIN DESCRIPTION:
BENNETT CREEK 82.0
END DESCRIPTION:
XS GIS Cut Line= 3
      2777105.64     10196103.12      2777822.82     10195883.34
      2778205.72     10196153.14
#Sta/Elev= 30
  4249.9 1343.87  4291.8 1343.31  4410.1 1335.79  4468.8 1332.73  4532.3 1328.30
  4544.0 1323.71  4571.6 1325.48  4576.8 1322.06  4604.3 1322.93  4609.5 1320.43
  4675.0 1319.19  4733.2 1319.89  4783.8 1322.61  4804.3 1328.99  4835.6 1324.83
  4896.6 1324.75  4952.8 1323.48  4989.5 1317.46  4990.0 1316.96  4995.5 1317.46
  5044.7 1319.37  5059.5 1321.46  5101.4 1320.29  5160.5 1326.94  5202.3 1326.41
  5246.7 1327.88  5346.0 1337.05  5368.6 1336.30  5382.7 1338.95  5468.4 1347.07
#Mann=7,-1,0
  4249.9    0.05       0  4410.1    0.12       0  4468.8    0.05       0
  4733.2    0.12       0  4896.6    0.05       0  4989.5    0.05       0
  4995.5    0.05       0
Bank Sta=4989.5,4995.5
Exp/Cntr=0.3,0.1

Type RM Length L Ch R = 1,40500,500,500,500
BEGIN DESCRIPTION:
BENNETT CREEK 81.0
END DESCRIPTION:
XS GIS Cut Line= 3
      2777253.21     10196351.51      2777746.11     10196331.77
      2778155.72     10196453.12
#Sta/Elev= 30
  4506.7 1331.53  4598.5 1327.56  4659.3 1326.32  4689.3 1328.84  4709.3 1328.07
  4759.4 1329.39  4809.4 1327.10  4829.4 1324.40  4838.0 1321.59  4843.0 1322.26
  4869.5 1320.09  4899.5 1322.12  4939.5 1322.44  4959.5 1320.08  4969.5 1317.82
  4979.6 1317.52  4993.5 1314.51  4994.0 1314.01  5001.1 1314.51  5010.0 1314.53
  5030.8 1320.49  5041.3 1321.54  5116.7 1323.23  5176.9 1325.04  5208.1 1327.92
  5228.7 1327.55  5260.3 1331.55  5364.6 1348.02  5416.7 1366.03  5427.2 1368.51
#Mann=5,-1,0
  4506.7    0.05       0  4598.5    0.12       0  4993.5    0.07       0
  5001.1    0.12       0  5116.7    0.05       0
Bank Sta=4993.5,5001.1
Exp/Cntr=0.3,0.1

Type RM Length L Ch R = 1,40000,500,500,500
BEGIN DESCRIPTION:
BENNETT CREEK 80.0
END DESCRIPTION:
XS GIS Cut Line= 3
      2777355.70     10196753.11      2777703.29     10196811.11
      2778105.71     10196603.10
#Sta/Elev= 30
  4647.6 1335.96  4718.4 1335.61  4840.2 1329.80  4880.8 1323.75  4911.2 1322.19
  4961.9 1315.44  4988.5 1314.30  4989.0 1313.80  4996.1 1314.30  5029.6 1314.71
  5051.7 1317.14  5068.2 1321.16  5166.4 1326.17  5196.3 1328.96  5251.0 1334.27
  5267.5 1337.67  5289.7 1338.30  5295.4 1340.35  5311.8 1341.42  5328.4 1345.66
  5334.0 1344.54  5350.5 1349.10  5356.1 1348.07  5372.6 1354.05  5378.3 1352.68
  5381.8 1354.38  5394.8 1361.00  5400.4 1360.06  5416.9 1366.44  5453.0 1369.76
#Mann=7,-1,0
  4647.6    0.12       0  4718.4    0.05       0  4988.5    0.05       0
  4996.1    0.05       0  5166.4    0.12       0  5196.3    0.05       0
  5381.8    0.12       0
Bank Sta=4988.5,4996.1
Exp/Cntr=0.3,0.1

Type RM Length L Ch R = 1,39500,500,500,500
BEGIN DESCRIPTION:
BENNETT CREEK 79.0
END DESCRIPTION:
XS GIS Cut Line= 3
      2777305.72     10197253.12      2777657.01     10197296.80
      2777905.64     10197403.09
#Sta/Elev= 30
  4646.0 1334.31  4706.4 1331.84  4716.5 1330.55  4726.6 1330.52  4744.8 1329.15
  4777.0 1327.44  4837.4 1325.97  4845.5 1325.20  4857.6 1322.47  4897.9 1319.86
  4938.2 1315.90  4948.3 1314.27  4961.6 1310.83  4968.4 1309.80  4988.6 1310.82
  5005.6 1309.61  5006.1 1309.11  5013.3 1309.61  5020.3 1312.25  5027.3 1313.88
  5042.1 1311.33  5050.9 1312.53  5056.3 1314.59  5074.4 1317.31  5079.9 1318.89
  5103.5 1321.90  5118.2 1324.77  5145.2 1326.26  5216.1 1332.55  5270.4 1335.69
#Mann=6,-1,0
  4646.0    0.12       0  4744.8    0.05       0  4961.6    0.12       0
  5005.6    0.07       0  5013.3    0.12       0  5145.2    0.05       0
Bank Sta=5005.6,5013.3
Exp/Cntr=0.3,0.1

Type RM Length L Ch R = 1,39000,500,500,500
BEGIN DESCRIPTION:
BENNETT CREEK 78.0
END DESCRIPTION:
XS GIS Cut Line= 3
      2777205.71     10197503.14      2777391.50     10197705.76
      2777655.64     10197803.09
#Sta/Elev= 30
  4725.1 1333.48  4760.5 1332.26  4774.7 1331.06  4788.9 1328.24  4857.8 1324.31
  4880.8 1320.80  4937.5 1315.40  4951.7 1312.91  4972.6 1307.90  5003.4 1306.46
  5004.4 1305.79  5004.9 1305.29  5012.1 1305.79  5033.4 1306.77  5047.6 1310.85
  5057.7 1312.38  5069.2 1315.54  5089.0 1318.07  5100.4 1320.80  5111.0 1321.57
  5119.4 1324.01  5124.8 1326.55  5143.0 1325.99  5155.2 1327.12  5183.2 1327.15
  5210.8 1326.98  5235.9 1329.85  5241.2 1329.51  5266.3 1332.22  5281.5 1332.84
#Mann=6,-1,0
  4725.1    0.12       0  4857.8    0.05       0  5004.4    0.05       0
  5012.1    0.05       0  5047.6    0.12       0  5183.2    0.05       0
Bank Sta=5004.4,5012.1
Exp/Cntr=0.3,0.1

Type RM Length L Ch R = 1,38500,500,500,500
BEGIN DESCRIPTION:
BENNETT CREEK 77.0
END DESCRIPTION:
XS GIS Cut Line= 3
      2776955.64     10198153.11      2777281.15     10198179.78
      2777705.66     10198003.12
#Sta/Elev= 30
  4673.4 1329.82  4723.6 1326.61  4753.7 1322.75  4773.8 1321.91  4834.0 1316.35
  4853.1 1313.33  4858.1 1313.89  4884.1 1311.90  4894.2 1309.86  4954.4 1302.37
  4994.5 1300.81  5003.4 1299.16  5003.9 1298.66  5011.2 1299.16  5015.7 1303.10
  5025.8 1305.15  5031.2 1304.81  5055.0 1306.88  5084.3 1306.54  5102.4 1307.26
  5113.5 1308.55  5243.6 1315.43  5297.4 1320.73  5329.8 1322.81  5339.0 1324.16
  5344.4 1323.97  5351.5 1325.82  5384.0 1328.25  5405.7 1331.01  5459.8 1333.79
#Mann=3,-1,0
  4673.4    0.05       0  5003.4    0.05       0  5011.2    0.05       0
Bank Sta=5003.4,5011.2
Exp/Cntr=0.3,0.1

Type RM Length L Ch R = 1,38000,500,500,500
BEGIN DESCRIPTION:
BENNETT CREEK 76.0
END DESCRIPTION:
XS GIS Cut Line= 3
      2776905.73     10198753.10      2777423.68     10198644.09
      2777805.69     10198153.10
#Sta/Elev= 30
  4470.7 1340.74  4501.3 1338.69  4590.1 1329.00  4664.8 1323.79  4695.5 1323.23
  4784.3 1314.30  4917.7 1303.60  4971.4 1296.67  5003.7 1294.21  5004.2 1293.71
  5015.2 1294.21  5015.8 1295.59  5024.0 1294.56  5030.3 1297.02  5038.4 1296.06
  5044.8 1298.85  5059.3 1298.46  5065.6 1301.73  5080.1 1303.52  5129.8 1303.83
  5144.5 1299.95  5152.5 1296.31  5166.0 1295.93  5173.3 1297.63  5272.8 1301.54
  5280.4 1303.88  5357.9 1314.76  5407.1 1319.47  5574.8 1328.66  5622.1 1331.20
#Mann=8,-1,0
  4470.7    0.05       0  4917.7    0.12       0  5003.7    0.07       0
  5015.2    0.12       0  5144.5    0.05       0  5280.4    0.12       0
  5407.1    0.05       0  5574.8    0.12       0
Bank Sta=5003.7,5015.2
Exp/Cntr=0.3,0.1

Type RM Length L Ch R = 1,37500,500,500,500
BEGIN DESCRIPTION:
BENNETT CREEK 75.0
END DESCRIPTION:
XS GIS Cut Line= 3
      2777155.68     10199053.11      2777361.52     10199127.01
      2777755.67     10199353.11
#Sta/Elev= 30
  4781.3 1316.36  4796.7 1316.04  4902.5 1304.84  4914.3 1303.29  4919.6 1303.43
  4951.3 1299.44  4961.9 1297.59  4970.5 1294.25  4983.2 1290.91  5000.6 1289.97
  5001.1 1289.47  5011.6 1289.47  5012.1 1289.97  5016.3 1292.02  5022.2 1296.08
  5050.9 1299.99  5065.4 1301.39  5131.6 1302.82  5204.9 1308.19  5263.8 1311.20
  5293.0 1314.29  5301.2 1314.48  5328.6 1319.44  5344.4 1320.98  5360.2 1323.68
  5366.0 1323.74  5381.8 1326.20  5419.2 1330.06  5431.4 1330.71  5454.4 1333.60
#Mann=4,-1,0
  4781.3    0.05       0  4902.5    0.12       0  5000.6    0.07       0
  5012.1    0.12       0
Bank Sta=5000.6,5012.1
Exp/Cntr=0.3,0.1

Type RM Length L Ch R = 1,37000,500,500,500
BEGIN DESCRIPTION:
BENNETT CREEK 74.0
END DESCRIPTION:
XS GIS Cut Line= 3
      2776655.65     10199403.10      2777163.57     10199580.49
      2777255.71     10199703.14
#Sta/Elev= 30
  4462.0 1328.65  4508.6 1325.54  4534.4 1322.73  4539.7 1323.30  4546.8 1322.01
  4589.1 1319.60  4632.8 1314.59  4684.3 1311.37  4695.1 1309.15  4720.7 1307.11
  4726.8 1306.03  4777.5 1302.21  4836.7 1300.22  4896.3 1299.16  4932.8 1296.70
  4938.7 1295.53  4949.3 1295.87  4958.5 1295.29  4970.5 1291.73  4989.6 1287.82
  4992.7 1285.45  4993.2 1284.95  5003.8 1284.95  5004.3 1285.45  5025.3 1292.41
  5031.5 1296.68  5053.3 1301.57  5075.3 1303.22  5114.0 1308.29  5153.4 1312.57
#Mann=5,-1,0
  4462.0    0.05       0  4836.7    0.12       0  4992.7    0.07       0
  5004.3    0.12       0  5114.0    0.05       0
Bank Sta=4992.7,5004.3
Exp/Cntr=0.3,0.1

Type RM Length L Ch R = 1,36500,500,500,500
BEGIN DESCRIPTION:
BENNETT CREEK 73.0
END DESCRIPTION:
XS GIS Cut Line= 3
      2776605.71     10199853.12      2776792.85     10199909.34
      2777055.72     10200003.12
#Sta/Elev= 30
  4804.6 1309.99  4815.0 1309.68  4826.3 1307.91  4846.3 1306.71  4859.4 1304.41
  4887.2 1302.52  4925.4 1297.16  4950.8 1294.66  4971.6 1287.56  4990.9 1283.69
  4991.4 1283.19  5002.0 1283.19  5002.5 1283.69  5004.2 1284.95  5013.6 1286.18
  5022.5 1289.21  5027.8 1291.56  5034.9 1292.87  5058.6 1295.75  5098.6 1296.90
  5120.2 1296.49  5140.4 1297.44  5145.7 1297.24  5162.3 1298.50  5176.6 1298.45
  5202.0 1300.03  5215.4 1300.12  5232.9 1301.96  5257.8 1303.01  5279.1 1305.56
#Mann=3,-1,0
  4804.6    0.12       0  4990.9    0.07       0  5002.5    0.12       0
Bank Sta=4990.9,5002.5
Exp/Cntr=0.3,0.1

Type RM Length L Ch R = 1,36000,500,500,500
BEGIN DESCRIPTION:
BENNETT CREEK 72.0
END DESCRIPTION:
XS GIS Cut Line= 3
      2776105.66     10200453.12      2776584.44     10200361.83
      2777580.98     10200372.34
#Sta/Elev= 30
  4512.6 1310.88  4624.6 1302.54  4716.2 1298.14  4757.5 1293.80  4767.1 1294.91
  4809.6 1292.74  4828.2 1290.87  4848.6 1285.48  4856.7 1284.82  4868.9 1288.29
  4892.2 1290.89  4930.0 1292.67  4950.4 1291.81  4966.1 1288.86  4971.1 1291.10
  4991.1 1286.77  4992.3 1281.92  4992.8 1281.42  5003.9 1281.92  5011.2 1283.10
  5041.2 1281.94  5081.2 1290.63  5091.3 1291.18  5181.3 1291.63  5289.8 1295.25
  5487.2 1296.03  5684.6 1298.48  5783.3 1300.05  5882.0 1301.36  5996.6 1303.00
#Mann=9,-1,0
  4512.6    0.05       0  4892.2    0.12       0  4992.3    0.07       0
  5003.9    0.12       0  5289.8    0.05       0  5487.2    0.12       0
  5684.6    0.05       0  5783.3    0.12       0  5882.0    0.05       0
Bank Sta=4992.3,5003.9
Exp/Cntr=0.3,0.1

Type RM Length L Ch R = 1,35500,500,500,500
BEGIN DESCRIPTION:
BENNETT CREEK 71.0
END DESCRIPTION:
XS GIS Cut Line= 3
      2776305.66     10200953.12      2776516.80     10200845.91
      2777477.24     10200736.92
#Sta/Elev= 30
  4763.2 1304.98  4821.7 1299.42  4838.3 1298.48  4843.9 1296.86  4852.9 1297.09
  4860.6 1296.22  4866.2 1294.71  4882.8 1293.97  4888.5 1292.74  4920.2 1291.40
  4942.7 1286.81  4949.6 1282.76  4955.2 1282.57  4971.9 1279.66  4987.5 1279.60
  4987.9 1279.05  4988.4 1278.55  5000.3 1279.05  5019.0 1280.26  5039.1 1288.71
  5049.2 1290.25  5099.5 1290.18  5200.2 1287.84  5220.3 1289.16  5340.4 1289.59
  5522.2 1290.71  5653.0 1294.20  5778.8 1299.11  5953.0 1308.05  5966.6 1308.15
#Mann=4,-1,0
  4763.2    0.05       0  4987.9    0.07       0  5000.3    0.05       0
  5340.4    0.05       0
Bank Sta=4987.9,5000.3
Exp/Cntr=0.3,0.1

Type RM Length L Ch R = 1,35000,500,500,500
BEGIN DESCRIPTION:
BENNETT CREEK 70.0
END DESCRIPTION:
XS GIS Cut Line= 3
      2776355.67     10201053.11      2776719.00     10201271.28
      2777105.66     10201653.09
#Sta/Elev= 30
  4576.2 1305.54  4692.9 1299.46  4816.7 1291.27  4918.2 1285.46  4933.8 1282.71
  4955.1 1281.28  4992.1 1274.51  5000.0 1275.09  5006.7 1273.22  5007.2 1272.72
  5019.4 1273.22  5020.2 1278.05  5027.2 1279.44  5034.3 1283.23  5041.4 1282.94
  5048.5 1284.90  5062.6 1286.23  5140.4 1286.20  5196.9 1284.47  5260.6 1285.60
  5295.9 1288.24  5310.1 1290.47  5317.2 1292.63  5331.3 1294.44  5375.6 1298.46
  5387.9 1300.62  5422.3 1303.66  5444.5 1306.06  5529.3 1310.50  5543.4 1312.11
#Mann=6,-1,0
  4576.2    0.05       0  4816.7    0.12       0  5006.7    0.07       0
  5019.4    0.12       0  5375.6    0.05       0  5422.3    0.12       0
Bank Sta=5006.7,5019.4
Exp/Cntr=0.3,0.1

Type RM Length L Ch R = 1,34500,500,500,500
BEGIN DESCRIPTION:
BENNETT CREEK 69.0
END DESCRIPTION:
XS GIS Cut Line= 3
      2776305.68     10201053.09      2776376.95     10201574.34
      2776755.66     10201953.08
#Sta/Elev= 30
  4473.9 1307.35  4504.2 1306.47  4582.3 1299.93  4701.4 1291.78  4796.9 1286.24
  4847.4 1281.89  4881.3 1278.16  4918.0 1277.37  4928.1 1278.09  4948.3 1276.48
  4968.5 1275.91  4988.7 1272.66  4990.5 1271.05  4991.0 1270.55  5003.3 1271.05
  5012.4 1272.77  5019.4 1272.87  5026.5 1278.99  5033.6 1275.53  5038.2 1278.48
  5040.7 1280.09  5047.7 1280.38  5083.1 1280.82  5111.4 1280.22  5139.7 1282.05
  5237.2 1284.03  5401.3 1288.19  5415.4 1289.36  5469.0 1291.39  5535.6 1293.70
#Mann=7,-1,0
  4473.9    0.05       0  4701.4    0.12       0  4990.5    0.07       0
  5003.3    0.12       0  5038.2    0.05       0  5237.2    0.12       0
  5469.0    0.05       0
Bank Sta=4990.5,5003.3
Exp/Cntr=0.3,0.1

Type RM Length L Ch R = 1,34000,500,500,500
BEGIN DESCRIPTION:
BENNETT CREEK 68.0
END DESCRIPTION:
XS GIS Cut Line= 3
      2775655.68     10201253.11      2776023.13     10201770.13
      2776955.70     10202403.12
#Sta/Elev= 30
  4365.7 1303.50  4587.1 1294.81  4667.0 1287.18  4702.7 1284.72  4717.5 1285.37
  4726.0 1283.72  4759.3 1281.11  4839.2 1277.72  4874.9 1277.38  4881.0 1278.23
  4967.1 1276.55  4975.7 1275.79  4992.4 1270.68  4992.9 1270.18  5005.2 1270.68
  5011.7 1271.41  5021.6 1274.16  5032.7 1276.14  5047.6 1276.59  5062.6 1275.69
  5116.1 1276.45  5208.5 1278.14  5365.1 1282.31  5514.8 1286.42  5529.7 1287.97
  5586.6 1289.00  5668.8 1292.56  5910.0 1303.47  6032.8 1311.13  6127.1 1313.52
#Mann=9,-1,0
  4365.7    0.05       0  4726.0    0.12       0  4992.4    0.07       0
  5005.2    0.12       0  5021.6    0.05       0  5116.1    0.12       0
  5208.5    0.05       0  5365.1    0.12       0  5668.8    0.05       0
Bank Sta=4992.4,5005.2
Exp/Cntr=0.3,0.1

Type RM Length L Ch R = 1,33500,500,500,500
BEGIN DESCRIPTION:
BENNETT CREEK 67.0
END DESCRIPTION:
XS GIS Cut Line= 3
      2775455.70     10202003.12      2775941.18     10202206.09
      2776355.68     10202303.11
#Sta/Elev= 30
  4473.8 1291.77  4565.2 1288.55  4679.7 1282.85  4712.2 1282.13  4755.6 1279.47
  4857.0 1275.67  4907.3 1273.44  4954.7 1272.85  4972.4 1271.21  4978.5 1268.31
  5018.8 1267.26  5019.3 1266.76  5031.6 1267.26  5035.4 1269.48  5045.7 1272.29
  5051.8 1272.94  5066.2 1272.57  5076.5 1271.19  5127.9 1274.15  5179.2 1274.46
  5189.5 1273.85  5210.0 1275.10  5232.0 1275.28  5240.8 1276.11  5269.3 1281.44
  5281.9 1286.03  5292.2 1288.04  5317.4 1291.14  5359.4 1293.90  5425.7 1295.16
#Mann=5,-1,0
  4473.8    0.05       0  4857.0    0.12       0  5018.8    0.07       0
  5031.6    0.12       0  5317.4    0.05       0
Bank Sta=5018.8,5031.6
Exp/Cntr=0.3,0.1

Type RM Length L Ch R = 1,33000,500,500,500
BEGIN DESCRIPTION:
BENNETT CREEK 66.0
END DESCRIPTION:
XS GIS Cut Line= 3
      2775455.69     10202203.12      2775655.42     10202534.71
      2776055.67     10202953.09
#Sta/Elev= 30
  4612.9 1288.85  4620.7 1287.35  4667.2 1283.16  4678.9 1281.62  4721.6 1279.95
  4737.2 1277.94  4752.7 1277.40  4764.7 1278.16  4779.9 1277.03  4795.4 1274.23
  4801.3 1274.56  4832.3 1271.60  4954.7 1270.55  4976.0 1268.83  4985.7 1266.04
  4991.6 1265.64  4996.1 1263.73  5006.6 1263.62  5007.1 1263.12  5019.5 1263.62
  5020.3 1265.36  5041.4 1267.86  5062.8 1267.60  5098.0 1269.03  5128.0 1272.14
  5218.5 1276.21  5260.7 1279.44  5331.4 1280.23  5472.9 1286.39  5579.0 1289.80
#Mann=5,-1,0
  4612.9    0.05       0  4667.2    0.12       0  5006.6    0.07       0
  5019.5    0.12       0  5128.0    0.05       0
Bank Sta=5006.6,5019.5
Exp/Cntr=0.3,0.1

Type RM Length L Ch R = 1,32500,281,281,281
BEGIN DESCRIPTION:
BENNETT CREEK 65.0
END DESCRIPTION:
XS GIS Cut Line= 3
      2774930.32     10201986.94      2775238.80     10202808.11
      2775655.69     10203203.11
#Sta/Elev= 30
  4122.8 1280.76  4214.9 1282.52  4300.3 1283.03  4374.7 1282.22  4380.1 1282.99
  4435.2 1281.84  4465.5 1282.63  4481.9 1281.59  4526.0 1282.13  4550.9 1281.58
  4575.8 1279.56  4661.1 1277.53  4666.5 1278.24  4721.6 1276.52  4746.5 1274.65
  4801.7 1273.45  4831.9 1271.47  4855.8 1271.59  4887.0 1270.38  4972.4 1265.13
  4977.5 1262.08  4978.0 1261.58  4990.4 1262.08  5000.0 1262.97  5015.5 1262.39
  5043.8 1265.48  5234.7 1268.82  5383.2 1274.89  5517.9 1282.05  5574.3 1283.81
#Mann=3,-1,0
  4122.8    0.05       0  4977.5    0.05       0  4990.4    0.05       0
Bank Sta=4977.5,4990.4
Exp/Cntr=0.3,0.1

Type RM Length L Ch R = 1,32219,719,719,719
BEGIN DESCRIPTION:
BENNETT CREEK 64.0
END DESCRIPTION:
XS GIS Cut Line= 3
      2774300.12     10202898.39      2775071.00     10203028.00
      2775655.71     10203303.12
#Sta/Elev= 30
  4218.3 1279.02  4305.1 1276.35  4325.3 1278.57  4345.6 1275.74  4355.8 1277.74
  4365.9 1277.80  4515.6 1273.93  4629.6 1272.64  4823.5 1263.92  4852.6 1263.59
  4879.0 1261.54  4944.7 1263.91  4984.5 1262.71  4994.6 1261.65  4998.6 1258.30
  4999.1 1257.80  5012.4 1258.30  5022.8 1261.38  5068.3 1265.69  5136.7 1264.79
  5171.0 1268.59  5193.4 1269.66  5256.2 1267.70  5307.4 1268.20  5324.6 1270.41
  5352.9 1270.20  5495.2 1278.24  5512.5 1277.94  5535.3 1280.21  5646.2 1284.19
#Mann=3,-1,0
  4218.3    0.05       0  4998.6    0.05       0  5012.4    0.05       0
Bank Sta=4998.6,5012.4
Exp/Cntr=0.3,0.1

Type RM Length L Ch R = 1,31500,500,500,500
BEGIN DESCRIPTION:
BENNETT CREEK 63.0
END DESCRIPTION:
XS GIS Cut Line= 3
      2774755.65     10203653.11      2775269.53     10203680.45
      2775655.66     10203353.13
#Sta/Elev= 30
  4485.4 1310.25  4545.5 1308.80  4565.5 1306.50  4575.0 1305.00  4605.6 1297.79
  4635.6 1292.91  4675.7 1285.28  4695.7 1280.48  4735.8 1273.52  4764.3 1270.40
  4769.3 1270.72  4845.9 1264.80  4926.1 1260.50  4958.5 1260.71  4979.6 1258.01
  4986.1 1256.46  4988.7 1254.47  4989.2 1253.97  5002.0 1253.97  5002.5 1254.47
  5023.4 1259.14  5031.1 1260.23  5045.4 1260.52  5059.7 1262.05  5094.8 1263.20
  5152.0 1263.74  5239.2 1266.98  5349.7 1272.73  5478.2 1282.33  5506.2 1283.71
#Mann=5,-1,0
  4485.4    0.05       0  4979.6    0.12       0  4988.7    0.07       0
  5002.5    0.12       0  5239.2    0.05       0
Bank Sta=4988.7,5002.5
Exp/Cntr=0.3,0.1

Type RM Length L Ch R = 1,31000,500,500,500
BEGIN DESCRIPTION:
BENNETT CREEK 62.0
END DESCRIPTION:
XS GIS Cut Line= 3
      2775005.68     10204053.11      2775517.42     10204108.16
      2775905.66     10203603.15
#Sta/Elev= 30
  4485.3 1281.90  4575.8 1277.84  4616.1 1274.42  4623.3 1273.02  4636.2 1273.44
  4686.5 1269.00  4736.8 1265.96  4904.4 1258.20  4958.0 1256.54  4978.1 1253.68
  4988.2 1253.49  4992.9 1252.64  4993.4 1252.14  5006.7 1252.64  5009.0 1255.26
  5017.2 1255.94  5023.5 1257.89  5058.9 1260.42  5094.7 1261.52  5107.7 1261.21
  5131.4 1261.59  5137.7 1260.95  5173.0 1261.10  5181.2 1260.35  5245.6 1260.44
  5359.7 1263.80  5467.6 1267.21  5531.4 1269.26  5579.9 1270.71  5637.0 1273.60
#Mann=7,-1,0
  4485.3    0.05       0  4992.9    0.05       0  5006.7    0.05       0
  5107.7    0.12       0  5359.7    0.05       0  5467.6    0.12       0
  5531.4    0.05       0
Bank Sta=4992.9,5006.7
Exp/Cntr=0.3,0.1

Type RM Length L Ch R = 1,30500,500,500,500
BEGIN DESCRIPTION:
BENNETT CREEK 61.0
END DESCRIPTION:
XS GIS Cut Line= 3
      2775405.65     10204803.14      2775773.03     10204531.50
      2776155.68     10204053.11
#Sta/Elev= 30
  4543.1 1271.12  4585.9 1269.32  4600.6 1269.55  4629.8 1268.42  4750.9 1266.03
  4829.2 1262.79  4892.8 1259.21  4907.4 1256.94  4951.3 1253.88  4972.1 1251.07
  4978.4 1249.69  4986.8 1250.06  4991.6 1248.89  4992.1 1248.39  5005.0 1248.39
  5005.5 1248.89  5014.7 1250.23  5022.7 1252.31  5029.1 1255.85  5036.4 1259.04
  5053.5 1259.07  5057.9 1259.17  5064.3 1258.36  5086.7 1258.87  5093.1 1257.79
  5118.7 1257.78  5164.4 1257.15  5299.6 1261.64  5427.7 1269.46  5612.6 1279.04
#Mann=5,-1,0
  4543.1    0.05       0  4991.6    0.03       0  5005.5    0.05       0
  5053.5    0.12       0  5118.7    0.05       0
Bank Sta=4991.6,5005.5
Exp/Cntr=0.3,0.1

Type RM Length L Ch R = 1,30000,500,500,500
BEGIN DESCRIPTION:
BENNETT CREEK 60.0
END DESCRIPTION:
XS GIS Cut Line= 3
      2775555.72     10205053.10      2776036.44     10204948.37
      2776455.68     10204603.12
#Sta/Elev= 30
  4508.0 1268.19  4630.8 1265.29  4682.0 1263.05  4712.7 1262.67  4804.8 1258.77
  4855.6 1255.80  4876.4 1255.57  4921.1 1256.55  4937.8 1256.34  4958.8 1253.10
  4968.5 1250.19  4978.8 1248.28  4982.0 1245.29  4982.5 1244.79  4995.4 1244.79
  4995.9 1245.29  4997.1 1247.09  5003.0 1247.97  5010.8 1247.99  5046.0 1256.33
  5060.3 1257.26  5066.8 1256.67  5081.1 1256.85  5089.0 1256.07  5095.5 1256.61
  5138.5 1255.40  5176.4 1255.67  5258.3 1259.65  5408.2 1263.57  5543.1 1269.03
#Mann=5,-1,0
  4508.0    0.05       0  4921.1    0.12       0  4982.0    0.07       0
  4995.9    0.12       0  5176.4    0.05       0
Bank Sta=4982,4995.9
Exp/Cntr=0.3,0.1

Type RM Length L Ch R = 1,29500,500,500,500
BEGIN DESCRIPTION:
BENNETT CREEK 59.0
END DESCRIPTION:
XS GIS Cut Line= 3
      2775855.69     10205753.10      2776349.31     10205332.06
      2777155.66     10205253.11
#Sta/Elev= 30
  4351.2 1267.52  4436.3 1265.34  4493.4 1261.90  4635.0 1256.49  4719.5 1254.52
  4883.2 1255.13  4932.6 1252.61  4940.3 1251.10  4946.8 1251.52  4973.8 1247.01
  4999.4 1245.17  4999.9 1244.67  5013.4 1245.17  5026.5 1246.97  5041.0 1251.32
  5046.6 1251.86  5066.7 1250.31  5106.9 1252.42  5137.0 1250.62  5187.4 1252.34
  5327.9 1254.09  5345.7 1252.10  5350.7 1253.42  5378.2 1250.56  5398.3 1249.80
  5447.2 1255.51  5452.3 1254.79  5548.8 1260.92  5559.0 1260.65  5810.2 1274.73
#Mann=5,-1,0
  4351.2    0.05       0  4973.8    0.12       0  4999.4    0.07       0
  5013.4    0.12       0  5187.4    0.05       0
Bank Sta=4999.4,5013.4
Exp/Cntr=0.3,0.1

Type RM Length L Ch R = 1,29000,500,500,500
BEGIN DESCRIPTION:
BENNETT CREEK 58.0
END DESCRIPTION:
XS GIS Cut Line= 3
      2775810.56     10205908.80      2776430.84     10205777.63
      2777255.82     10205874.08
#Sta/Elev= 30
  4366.0 1270.30  4381.5 1268.58  4432.6 1265.88  4462.1 1262.95  4467.2 1263.81
  4511.8 1259.72  4516.9 1260.29  4575.7 1257.21  4596.1 1257.35  4626.8 1255.90
  4755.3 1253.73  4760.4 1254.39  4805.0 1251.30  4831.2 1251.20  4841.4 1249.72
  4923.2 1247.68  4949.0 1244.96  4993.7 1244.84  4994.2 1243.36  4994.7 1242.86
  5009.9 1243.36  5010.9 1243.50  5035.1 1246.89  5055.2 1245.48  5109.8 1246.92
  5216.3 1250.95  5345.4 1251.79  5508.3 1254.37  5528.4 1255.49  5830.6 1262.10
#Mann=5,-1,0
  4366.0    0.05       0  4994.2    0.05       0  5009.9    0.05       0
  5010.9    0.12       0  5109.8    0.05       0
Bank Sta=4994.2,5009.9
Exp/Cntr=0.3,0.1

Type RM Length L Ch R = 1,28500,500,500,500
BEGIN DESCRIPTION:
BENNETT CREEK 57.0
END DESCRIPTION:
XS GIS Cut Line= 3
      2775805.67     10206053.11      2776281.43     10206250.55
      2776805.70     10206603.12
#Sta/Elev= 30
  4484.9 1267.60  4560.7 1263.35  4582.4 1261.06  4605.9 1259.90  4653.6 1256.10
  4712.3 1253.56  4730.6 1251.88  4777.2 1249.41  4783.8 1248.45  4813.1 1248.22
  4820.5 1247.41  4919.4 1244.06  4961.3 1241.96  4967.1 1241.13  4991.0 1240.71
  4991.7 1239.18  4992.2 1238.68  5006.9 1238.68  5007.4 1239.18  5027.3 1240.82
  5033.4 1240.07  5069.4 1241.34  5113.6 1244.34  5243.3 1247.29  5249.3 1248.18
  5285.3 1248.50  5351.3 1252.15  5444.3 1254.96  5588.3 1261.59  5631.8 1264.70
#Mann=3,-1,0
  4484.9    0.05       0  4991.7    0.05       0  5007.4    0.05       0
Bank Sta=4991.7,5007.4
Exp/Cntr=0.3,0.1

Type RM Length L Ch R = 1,28000,500,500,500
BEGIN DESCRIPTION:
BENNETT CREEK 56.0
END DESCRIPTION:
XS GIS Cut Line= 3
      2775555.69     10206353.12      2776041.70     10206680.53
      2776855.67     10206753.11
#Sta/Elev= 30
  4414.0 1276.13  4463.5 1272.76  4493.4 1269.05  4550.4 1264.10  4558.7 1264.23
  4580.4 1261.43  4637.4 1257.21  4667.2 1256.27  4673.4 1254.95  4694.4 1254.56
  4709.4 1252.70  4745.3 1251.55  4760.3 1249.91  4976.2 1241.95  4991.2 1240.05
  4991.5 1234.56  4992.0 1234.06  5007.3 1234.56  5014.0 1236.32  5044.2 1237.92
  5054.2 1236.90  5087.4 1238.90  5114.4 1238.88  5174.7 1242.38  5295.2 1244.35
  5355.4 1246.47  5636.5 1259.12  5656.6 1258.88  5706.8 1260.98  5817.2 1266.48
#Mann=3,-1,0
  4414.0    0.05       0  4991.5    0.03       0  5007.3    0.05       0
Bank Sta=4991.5,5007.3
Exp/Cntr=0.3,0.1

Type RM Length L Ch R = 1,27500,500,500,500
BEGIN DESCRIPTION:
BENNETT CREEK 55.0
END DESCRIPTION:
XS GIS Cut Line= 3
      2775605.68     10207103.11      2775949.25     10207167.77
      2776778.44     10207501.70
#Sta/Elev= 30
  4650.4 1255.36  4772.5 1250.73  4823.4 1246.91  4839.1 1244.05  4844.2 1245.52
  4891.6 1239.16  4896.7 1240.65  4915.0 1237.92  5017.2 1236.14  5017.7 1235.64
  5033.6 1236.14  5103.3 1237.06  5210.7 1239.93  5216.1 1240.94  5240.3 1240.32
  5269.8 1242.06  5294.0 1241.80  5299.4 1242.88  5318.2 1242.37  5323.6 1243.44
  5347.7 1242.87  5353.1 1243.98  5395.0 1244.46  5508.9 1249.30  5538.4 1249.14
  5562.6 1250.79  5568.0 1249.96  5586.8 1250.92  5707.7 1250.92  5893.9 1253.34
#Mann=3,-1,0
  4650.4    0.05       0  5017.2    0.03       0  5033.6    0.05       0
Bank Sta=5017.2,5033.6
Exp/Cntr=0.3,0.1

Type RM Length L Ch R = 1,27000,500,500,500
BEGIN DESCRIPTION:
BENNETT CREEK 54.0
END DESCRIPTION:
XS GIS Cut Line= 3
      2775455.66     10207303.10      2775962.83     10207664.56
      2776355.66     10207603.12
#Sta/Elev= 30
  4377.2 1256.76  4607.1 1246.86  4657.5 1245.74  4693.2 1244.01  4714.1 1244.28
  4821.0 1241.06  4900.9 1235.70  4921.8 1234.77  4942.7 1235.05  4957.5 1233.51
  4966.1 1231.26  4972.2 1232.67  4978.8 1228.98  4979.3 1228.48  4995.2 1228.98
  4998.7 1230.22  5023.1 1230.93  5040.0 1235.32  5045.1 1234.90  5057.9 1236.22
  5073.7 1237.54  5120.2 1239.04  5205.3 1242.47  5233.2 1244.34  5245.8 1244.25
  5296.0 1247.35  5301.0 1246.89  5363.7 1252.44  5368.8 1251.83  5397.6 1254.39
#Mann=5,-1,0
  4377.2    0.05       0  4978.8    0.05       0  4995.2    0.05       0
  5057.9    0.12       0  5120.2    0.05       0
Bank Sta=4978.8,4995.2
Exp/Cntr=0.3,0.1

Type RM Length L Ch R = 1,26500,500,500,500
BEGIN DESCRIPTION:
BENNETT CREEK 53.0
END DESCRIPTION:
XS GIS Cut Line= 3
      2775505.69     10207553.13      2775694.60     10208038.14
      2775955.69     10208303.12
#Sta/Elev= 30
  4479.5 1249.47  4489.0 1249.96  4494.4 1249.19  4518.9 1248.81  4543.4 1247.01
  4554.6 1247.17  4711.9 1240.32  4771.7 1238.59  4780.0 1237.04  4790.7 1238.02
  4805.8 1237.70  4887.3 1234.33  4905.0 1234.46  4919.5 1233.04  4929.5 1233.67
  4940.9 1233.29  4964.7 1231.31  4983.9 1227.31  4994.6 1228.64  5003.1 1225.98
  5003.6 1225.48  5019.0 1225.48  5019.5 1225.98  5027.2 1227.97  5039.6 1230.09
  5067.9 1236.60  5117.5 1242.27  5315.5 1257.19  5329.6 1257.37  5372.0 1260.24
#Mann=5,-1,0
  4479.5    0.05       0  4805.8    0.12       0  5003.1    0.07       0
  5019.5    0.12       0  5027.2    0.05       0
Bank Sta=5003.1,5019.5
Exp/Cntr=0.3,0.1

Type RM Length L Ch R = 1,26000,500,500,500
BEGIN DESCRIPTION:
BENNETT CREEK 52.0
END DESCRIPTION:
XS GIS Cut Line= 3
      2775305.68     10207553.11      2775205.58     10208076.63
      2775455.69     10208453.12
#Sta/Elev= 30
  4467.0 1253.16  4545.1 1250.05  4550.2 1250.47  4597.2 1247.16  4602.3 1248.17
  4706.4 1241.12  4731.7 1240.38  4782.6 1237.19  4945.5 1231.70  4971.9 1229.84
  4977.0 1230.44  4986.2 1229.07  4997.3 1224.45  4997.8 1223.95  5013.8 1224.45
  5019.8 1225.49  5068.6 1226.40  5077.7 1228.54  5087.7 1229.26  5140.8 1231.02
  5192.2 1236.38  5243.0 1240.24  5294.1 1242.68  5300.1 1242.12  5307.9 1243.40
  5315.2 1243.19  5321.2 1244.30  5351.3 1246.36  5380.0 1246.97  5452.0 1251.84
#Mann=5,-1,0
  4467.0    0.05       0  4997.3    0.05       0  5013.8    0.05       0
  5087.7    0.12       0  5192.2    0.05       0
Bank Sta=4997.3,5013.8
Exp/Cntr=0.3,0.1

Type RM Length L Ch R = 1,25500,500,500,500
BEGIN DESCRIPTION:
BENNETT CREEK 51.0
END DESCRIPTION:
XS GIS Cut Line= 3
      2774605.68     10208103.10      2774790.27     10208281.63
      2775205.69     10208703.12
#Sta/Elev= 30
  4743.2 1244.59  4813.8 1238.94  4856.3 1237.17  4950.3 1229.41  4983.6 1225.41
  4990.8 1222.05  4996.5 1220.71  4997.0 1220.21  5012.6 1220.21  5013.1 1220.71
  5019.0 1222.97  5026.1 1224.38  5040.3 1224.83  5047.3 1226.84  5054.4 1226.85
  5061.4 1227.79  5103.9 1226.44  5132.1 1227.30  5139.3 1228.15  5146.3 1227.91
  5155.7 1228.82  5181.7 1230.22  5210.0 1230.29  5273.6 1232.31  5316.0 1234.71
  5358.4 1235.27  5507.0 1244.77  5549.4 1246.80  5570.6 1248.59  5591.8 1248.65
#Mann=5,-1,0
  4743.2    0.05       0  4950.3    0.12       0  4996.5    0.07       0
  5013.1    0.12       0  5155.7    0.05       0
Bank Sta=4996.5,5013.1
Exp/Cntr=0.3,0.1

Type RM Length L Ch R = 1,25000,500,500,500
BEGIN DESCRIPTION:
BENNETT CREEK 50.0
END DESCRIPTION:
XS GIS Cut Line= 3
      2774455.69     10208253.14      2774495.37     10208620.00
      2774905.68     10208853.11
#Sta/Elev= 30
  4631.0 1242.71  4676.8 1238.12  4701.4 1237.26  4791.9 1231.00  4875.0 1226.72
  4882.4 1225.93  4942.8 1224.72  4957.1 1223.20  4974.3 1222.45  4983.0 1219.64
  4993.1 1218.56  4999.1 1216.92  5008.7 1216.77  5009.2 1216.27  5025.3 1216.77
  5054.5 1219.73  5060.3 1222.58  5097.8 1228.79  5113.6 1229.57  5119.4 1228.73
  5159.6 1230.61  5161.4 1230.68  5184.4 1231.81  5194.4 1231.55  5200.1 1232.44
  5230.4 1233.65  5237.6 1234.71  5253.4 1234.78  5318.4 1238.14  5471.9 1243.15
#Mann=7,-1,0
  4631.0    0.05       0  4875.0    0.12       0  4974.3    0.05       0
  5008.7    0.03       0  5025.3    0.05       0  5159.6    0.12       0
  5161.4    0.05       0
Bank Sta=5008.7,5025.3
Exp/Cntr=0.3,0.1
