HEC-RAS study HICKORY CREEK.prj: HICKORY CREEK Base Level Engineering

--- HICKORY CREEK.g01 (geometry) --- (continued)

Type RM Length L Ch R = 1 ,43000   ,500,500,500
BEGIN DESCRIPTION:
HICKORY CREEK 86.0
END DESCRIPTION:
XS GIS Cut Line= 4
      2753447.73      10205500.4      2753796.53     10205066.01
      2753927.45     10204490.23      2753587.61     10204041.59
#Sta/Elev= 30
  4442.9 1256.56  4531.5  1253.9  4595.6 1248.31  4603.5 1246.13  4609.9  1247.2
  4638.7 1243.37  4723.6 1237.19  4745.9  1232.9  4752.4 1233.24  4766.8 1228.77
  4773.2 1229.37  4781.2 1226.36  4787.6    1226    4810 1216.99  4824.2 1214.32
  4909.2 1207.52  4973.2 1207.71  5034.3 1206.78  5035.8 1205.78  5113.8 1205.78
  5115.3 1206.78  5115.8 1213.73  5167.6 1221.56  5195.9 1225.75  5292.3  1223.5
  5377.6 1226.64  5577.3 1236.98  5761.8 1240.94  6017.7 1241.28  6153.3 1244.01
#Mann= 4 ,-1 , 0
  4442.9     .05       0  4973.2     .05       0  5167.6     .12       0
  5377.6     .05       0
Bank Sta=5034.3,5115.3
XS Rating Curve= 0 ,0
Exp/Cntr=0.3,0.1

Type RM Length L Ch R = 1 ,42500   ,500,500,500
BEGIN DESCRIPTION:
HICKORY CREEK 85.0
END DESCRIPTION:
XS GIS Cut Line= 4
      2753467.69     10205620.35      2753797.43     10205585.38
      2754188.52     10205363.77      2754605.72     10205003.08
#Sta/Elev= 30
  4218.9 1254.65  4291.9 1249.67  4347.6 1241.29  4391.7 1242.95  4438.1 1241.99
  4518.6 1230.06  4705.4 1222.51  4770.3  1216.9  4829.1 1212.91  4845.4 1210.64
  4858.8 1206.42  4894.4 1206.01  4916.3 1208.03  4926.2 1205.91  4971.9 1205.24
  4973.4 1204.24  5052.9 1205.24  5104.5 1207.27    5133 1212.93  5154.9 1214.67
  5182.4 1207.18  5196.6 1207.42  5239.4 1218.02  5302.5 1226.54  5345.2 1235.14
  5402.8 1247.93  5431.3 1250.22  5452.2    1249  5466.4 1251.55  5551.5 1255.46
#Mann= 9 ,-1 , 0
  4218.9     .05       0  4291.9     .12       0  4391.7     .05       0
  4770.3     .12       0  4829.1     .05       0  4971.9     .03       0
  5052.9     .05       0  5302.5     .12       0  5345.2     .05       0
Bank Sta=4971.9,5052.9
XS Rating Curve= 0 ,0
Exp/Cntr=0.3,0.1

Type RM Length L Ch R = 1 ,42000   ,500,500,500
BEGIN DESCRIPTION:
HICKORY CREEK 84.0
END DESCRIPTION:
XS GIS Cut Line= 4
      2753252.81     10206149.94      2753915.46     10206102.07
      2754426.67     10205771.23      2754805.66     10205253.15
#Sta/Elev= 30
  3726.7 1245.76  3859.9 1237.49  3945.2 1234.52  4120.6 1231.96  4190.8 1232.44
  4331.1 1228.96    4413 1230.11  4558.1 1229.16  4745.4 1219.78  4781.7 1219.09
  4860.2 1212.85  4890.5 1211.74  4903.5 1209.59  4911.6 1206.93  4913.1 1203.92
  4914.6 1202.92    4993 1202.92  4994.5 1203.92    5134 1206.95  5162.1 1204.52
  5176.7 1204.69  5277.1 1213.39  5319.8 1220.31  5406.5 1228.38    5413  1230.2
  5442.3 1233.18  5448.5 1235.11  5456.1 1234.67  5492.5 1236.78  5641.9 1246.17
#Mann= 5 ,-1 , 0
  3726.7     .12       0  3945.2     .05       0  4913.1     .05       0
  4994.5     .05       0  5492.5     .05       0
Bank Sta=4913.1,4994.5
XS Rating Curve= 0 ,0
Exp/Cntr=0.3,0.1

Type RM Length L Ch R = 1 ,41500   ,500,500,500
BEGIN DESCRIPTION:
HICKORY CREEK 83.0
END DESCRIPTION:
XS GIS Cut Line= 5
      2753257.85     10206219.89      2754260.89      10206289.9
      2754681.53     10206189.23      2754996.51     10206124.96
       2755780.8     10206139.95
#Sta/Elev= 30
    3562 1247.11  3569.9 1246.91    3640 1239.63  3890.6 1229.56  4113.6  1227.6
  4361.8 1234.26    4442 1232.13  4660.5 1219.68  4749.7  1217.2  4833.8 1208.21
    4850 1203.91  4973.7 1202.45  4975.2 1201.45  5055.1 1202.45    5058 1204.68
  5065.5 1205.77  5187.9 1211.47  5249.2 1217.77  5269.6 1219.69  5350.6 1220.96
  5460.7 1215.99  5491.1 1212.06  5520.7 1213.99  5540.7 1217.46  5590.7 1218.24
  5660.7 1223.25  5880.7 1232.78  6007.8 1243.01  6012.8 1241.75  6105.9 1251.96
#Mann= 5 ,-1 , 0
    3562     .12       0  3569.9     .05       0  4973.7     .05       0
  5249.2     .05       0  5590.7     .05       0
Bank Sta=4973.7,5055.1
XS Rating Curve= 0 ,0
Exp/Cntr=0.3,0.1

Type RM Length L Ch R = 1 ,41000   ,500,500,500
BEGIN DESCRIPTION:
HICKORY CREEK 82.0
END DESCRIPTION:
XS GIS Cut Line= 4
      2753247.89     10206329.81      2754142.17      10206594.6
      2754686.29     10206669.45      2755121.06     10206674.53
#Sta/Elev= 30
  3518.1 1243.17  3584.6 1238.89  3766.1 1229.58  3943.4 1224.15  4041.5 1221.25
  4099.8  1222.5    4152 1221.34  4308.4 1227.68  4339.7 1231.76  4422.9 1235.94
  4433.6 1237.56  4514.9 1236.81  4694.1 1220.27  4771.2 1215.45  4848.2 1207.62
  4878.3  1202.7  4888.4 1203.47  4938.4 1200.79  4939.9 1199.79  5018.4 1199.79
  5019.9 1200.79  5089.4  1205.9  5139.4 1206.64  5159.4 1211.36  5179.4 1220.29
  5219.4 1230.78  5299.4  1245.7  5339.4 1250.85  5369.4 1252.64  5434.8 1254.27
#Mann= 6 ,-1 , 0
  3518.1     .12       0  3584.6     .05       0  3943.4     .05       0
  4938.4     .03       0  5019.9     .05       0  5369.4     .05       0
Bank Sta=4938.4,5019.9
XS Rating Curve= 0 ,0
Exp/Cntr=0.3,0.1

Type RM Length L Ch R = 1 ,40500   ,500,500,500
BEGIN DESCRIPTION:
HICKORY CREEK 81.0
END DESCRIPTION:
XS GIS Cut Line= 4
      2753777.46     10207339.02      2754655.11     10207146.62
       2755001.5     10207074.23      2755156.39     10206849.38
#Sta/Elev= 30
  4101.5  1249.4  4161.1 1243.32  4345.4 1226.12  4560.4 1212.36  4574.2 1209.96
  4601.3 1216.39  4759.8 1215.96  4808.7 1212.79  4867.5  1205.4  4896.4 1200.52
    4970 1199.68  4971.5 1198.68  5051.5 1199.68  5088.9 1204.57  5153.8 1204.97
  5183.8 1207.86  5233.8 1220.74  5245.8 1221.95  5333.7 1226.76  5401.5 1227.56
  5473.2 1233.05  5494.2 1233.56    5509 1235.95  5515.1 1234.87  5523.9 1236.33
    5530 1234.97  5544.9 1236.96  5565.8  1236.5  5595.6 1239.74  5626.9 1240.71
#Mann= 5 ,-1 , 0
  4101.5     .05       0  4161.1     .05       0  4867.5     .03       0
  5051.5     .05       0  5473.2     .05       0
Bank Sta=4970,5051.5
XS Rating Curve= 0 ,0
Exp/Cntr=0.3,0.1

Type RM Length L Ch R = 1 ,40000   ,500,500,500
BEGIN DESCRIPTION:
HICKORY CREEK 80.0
END DESCRIPTION:
XS GIS Cut Line= 3
      2754032.28      10208113.4      2754741.82     10207618.65
      2755486.08     10207513.89
#Sta/Elev= 30
    4135 1235.43  4216.3 1229.62  4237.2 1230.28  4266.9 1227.51  4281.7 1228.84
  4287.8 1226.32  4296.6 1227.87  4302.7  1225.2  4317.5 1225.31    4389 1219.09
  4496.4 1213.11  4561.8 1214.82  4704.9 1214.58  4740.6 1210.62  4755.5 1207.52
  4812.2 1203.23  4841.9  1199.2  4878.7 1197.95  4880.2 1196.95  4960.3 1197.95
  4970.1 1199.27    5014 1198.77  5104.9 1204.16  5205.9 1205.74  5266.5 1208.44
  5362.5 1217.63  5417.9 1220.64  5433.7 1223.34  5640.1 1231.95  5751.6 1236.64
#Mann= 5 ,-1 , 0
    4135     .05       0  4216.3     .05       0  4878.7     .03       0
  4960.3     .05       0  5640.1     .05       0
Bank Sta=4878.7,4960.3
XS Rating Curve= 0 ,0
Exp/Cntr=0.3,0.1

Type RM Length L Ch R = 1 ,39500   ,500,500,500
BEGIN DESCRIPTION:
HICKORY CREEK 79.0
END DESCRIPTION:
XS GIS Cut Line= 3
      2754396.97     10208463.15      2754832.65     10208081.05
      2755496.13     10207663.76
#Sta/Elev= 30
  4420.5  1229.4    4590 1222.09  4610.9 1222.39  4625.1 1220.91  4631.8 1221.87
  4639.4 1220.05    4646  1221.2  4653.6 1218.05  4788.4 1209.61  4816.8 1202.04
  4823.5  1202.8  4837.7 1207.32  4901.3 1204.21  4923.1 1199.85  4924.1 1197.02
  4925.6 1196.02  5004.2 1196.02  5005.7 1197.02  5022.8 1197.81  5059.3 1197.38
  5174.7 1201.24  5211.2 1198.55  5217.1 1200.33  5239.9 1202.23  5334.4 1204.66
  5363.1 1208.99  5405.6 1212.71  5509.2 1217.59  5609.3 1224.74  5783.8 1234.41
#Mann= 4 ,-1 , 0
  4420.5     .05       0  4925.6    .035       0  5022.8     .05       0
  5609.3     .05       0
Bank Sta=4924.1,5005.7
XS Rating Curve= 0 ,0
Exp/Cntr=0.3,0.1

Type RM Length L Ch R = 1 ,39000   ,500,500,500
BEGIN DESCRIPTION:
HICKORY CREEK 78.0
END DESCRIPTION:
XS GIS Cut Line= 3
      2754905.69     10208853.11      2755127.37     10208461.04
      2755505.67     10207953.14
#Sta/Elev= 30
  4549.6 1233.44  4579.2 1231.66  4622.5 1224.56    4630 1221.19  4644.1 1218.05
  4697.6 1210.71    4725 1212.08  4778.4 1202.03  4784.2 1203.99  4790.8 1201.34
    4812    1202  4821.7 1204.18  4827.5 1202.31  4843.4 1206.78    4865 1206.59
  4924.2 1202.44  4945.8 1199.61  4955.1 1195.85  4956.6 1194.85  5035.2 1194.85
  5036.7 1195.85    5184 1199.83    5234 1197.79  5290.3 1198.57  5311.1 1197.49
  5374.5 1206.19  5446.7 1212.58  5533.6 1217.79  5611.9 1224.17  5633.3 1225.23
#Mann= 6 ,-1 , 0
  4549.6     .05       0    4812     .05       0  4955.1    .035       0
  5036.7     .05       0  5374.5     .05       0  5611.9     .05       0
Bank Sta=4955.1,5036.7
XS Rating Curve= 0 ,0
Exp/Cntr=0.3,0.1

Type RM Length L Ch R = 1 ,38500   ,500,500,500
BEGIN DESCRIPTION:
HICKORY CREEK 77.0
END DESCRIPTION:
XS GIS Cut Line= 3
      2755251.29     10209177.63      2755570.38     10208656.93
      2755990.69     10207968.61
#Sta/Elev= 30
  4389.3 1222.65    4431 1219.24  4620.6 1211.67  4651.4 1212.06  4715.3 1208.72
  4730.7 1209.88  4773.3  1207.3  4810.1 1208.86  4825.5 1206.59  4831.4 1207.53
  4846.8 1204.06  4852.7  1205.5  4862.2 1203.42  4868.1 1205.27  4875.5 1200.31
  4883.5 1198.86  4934.1 1195.97  4958.5 1192.57    4960 1191.57  5040.1 1192.57
  5042.2 1196.19  5086.5 1194.19  5131.2 1196.19  5189.3 1195.08  5274.5 1196.59
  5311.3 1203.12  5332.6 1204.31  5625.5 1215.24  5727.4 1221.73  5806.5 1223.84
#Mann= 3 ,-1 , 0
  4389.3     .05       0  4958.5     .03       0  5040.1     .05       0
Bank Sta=4958.5,5040.1
XS Rating Curve= 0 ,0
Exp/Cntr=0.3,0.1

Type RM Length L Ch R = 1 ,38000   ,500,500,500
BEGIN DESCRIPTION:
HICKORY CREEK 76.0
END DESCRIPTION:
XS GIS Cut Line= 3
      2755645.99     10209452.42      2755995.02       10208877.
      2756335.45     10208243.36
#Sta/Elev= 30
    4327 1230.34  4328.7 1230.34  4450.4  1217.6  4582.2 1213.71    4683 1205.47
    4778 1200.65  4829.1 1201.37  4857.5 1197.32    4873 1198.92  4878.8 1197.18
  4894.3 1197.93  4900.2 1195.67  4922.7  1196.4  4999.3 1189.17  5027.1 1190.72
  5054.9 1189.14  5071.1 1191.85  5136.9 1193.28  5227.5 1188.34    5229 1187.34
  5309.2 1188.34  5312.2 1195.07  5350.3 1197.11  5394.2 1203.29  5410.4 1209.09
  5416.1 1206.56  5432.3 1211.58  5498.1  1215.9  5514.3 1213.79  5719.3 1223.83
#Mann= 4 ,-1 , 0
    4327     .12       0  4328.7     .05       0  5227.5     .03       0
  5309.2     .05       0
Bank Sta=5227.5,5309.2
XS Rating Curve= 0 ,0
Exp/Cntr=0.3,0.1

Type RM Length L Ch R = 1 ,37500   ,500,500,500
BEGIN DESCRIPTION:
HICKORY CREEK 75.0
END DESCRIPTION:
XS GIS Cut Line= 3
      2756025.71     10209667.22      2756420.87     10209091.85
      2756390.43     10208288.33
#Sta/Elev= 30
    4302  1227.5  4309.9  1227.4  4428.3 1222.65  4506.1 1215.93    4521 1213.02
  4537.4 1213.24  4653.2 1205.91  4682.3 1203.32  4715.2 1204.17  4721.3 1201.89
    4772 1195.63  4837.7 1190.28  4873.6 1191.34  4930.4 1189.33  4987.2 1184.35
  5098.8 1190.94  5148.8 1187.64  5178.9 1187.83  5188.9 1189.73  5238.1 1184.08
  5239.6 1183.08  5319.8 1184.08    5329 1194.86    5339 1197.82  5440.4 1207.91
  5514.4  1214.4  5549.1 1217.03  5579.2 1214.28  5619.2 1215.09  5804.1 1222.67
#Mann= 9 ,-1 , 0
    4302     .05       0  4309.9     .12       0  4537.4     .05       0
  4653.2     .12       0  4682.3     .05       0  5238.1     .03       0
  5319.8     .05       0  5440.4     .12       0  5514.4     .05       0
Bank Sta=5238.1,5319.8
XS Rating Curve= 0 ,0
Exp/Cntr=0.3,0.1

Type RM Length L Ch R = 1 ,37000   ,343,343,343
BEGIN DESCRIPTION:
HICKORY CREEK 74.0
END DESCRIPTION:
XS GIS Cut Line= 4
       2756060.7      10209682.2      2756204.61     10209586.53
      2756602.75     10209519.79      2757409.67     10209387.44
#Sta/Elev= 30
  4423.5 1225.94  4499.3 1222.68  4505.3 1224.09  4520.4 1221.57  4568.3 1220.14
  4599.4    1218  4645.1 1210.79  4650.2 1211.82  4678.5 1206.88    4724  1202.4
  4800.2 1196.29  4871.2 1185.18  4911.7 1189.36  4948.4 1182.83  5022.9 1179.49
  5024.4 1178.49  5104.7 1179.49  5131.8 1185.55  5136.9 1184.51  5175.2 1188.08
  5193.1 1183.36    5236  1189.9  5266.4 1191.08  5337.4 1204.15    5382 1204.15
    5571 1214.33  5688.5 1231.11  5732.6 1229.58  5768.9 1231.84  5817.7 1233.59
#Mann= 6 ,-1 , 0
  4423.5     .05       0  4568.3     .12       0    4724     .05       0
  5022.9     .03       0  5104.7     .05       0  5768.9     .12       0
Bank Sta=5022.9,5104.7
XS Rating Curve= 0 ,0
Exp/Cntr=0.3,0.1

Type RM Length L Ch R = 1 ,36657   ,657,657,657
BEGIN DESCRIPTION:
HICKORY CREEK 73.0
END DESCRIPTION:
XS GIS Cut Line= 3
      2755965.75     10209902.04      2756612.25       10209861.
      2757580.85     10209628.13
#Sta/Elev= 30
  4352.2 1228.98  4410.7 1222.41  4415.8 1223.37  4569.8 1211.79  4574.8 1212.72
  4742.9 1201.31    4803 1199.26  4843.1 1195.86  4913.3 1186.31  4963.4 1184.72
  4993.4  1178.2  5034.4 1179.55  5057.6 1179.25  5058.7 1177.43  5060.2 1176.43
  5140.5 1177.43  5147.5  1178.9  5157.8 1177.51  5183.5 1181.15  5188.7 1183.31
  5225.5 1187.91  5351.3 1196.12  5529.5 1215.44  5608.2 1215.34  5744.4 1221.85
  5781.2 1221.52  5836.6  1226.9    5888 1228.88  5925.4 1232.18  5996.2 1239.28
#Mann= 4 ,-1 , 0
  4352.2     .05       0  5058.7     .03       0  5140.5     .05       0
  5925.4     .12       0
Bank Sta=5058.7,5140.5
XS Rating Curve= 0 ,0
Exp/Cntr=0.3,0.1

Type RM Length L Ch R = 1 ,36000   ,500,500,500
BEGIN DESCRIPTION:
HICKORY CREEK 72.0
END DESCRIPTION:
XS GIS Cut Line= 3
      2755925.76     10210386.67      2756793.18     10210457.43
       2757359.7     10210436.63
#Sta/Elev= 30
  4129.7 1220.51  4151.1 1218.11  4280.1 1212.38  4410.6 1209.66  4516.2 1204.67
    4551 1204.06  4637.9 1196.53  4642.9 1197.15  4691.5 1194.02  4741.7 1189.14
  4821.9    1184    4862 1178.09  4932.3 1177.83  4957.8 1176.14  4959.3 1175.14
  5038.2 1175.14  5039.7 1176.14  5062.5 1181.12  5082.6 1182.88  5122.6 1190.22
  5142.6 1190.35  5212.6 1196.67  5222.7 1198.75  5255.8 1198.95  5262.7 1200.12
  5342.7 1204.35  5392.8 1214.37  5442.8 1218.62  5532.9 1223.88  5566.9 1224.53
#Mann= 3 ,-1 , 0
  4129.7     .05       0  4957.8     .03       0  5039.7     .05       0
Bank Sta=4957.8,5039.7
XS Rating Curve= 0 ,0
Exp/Cntr=0.3,0.1

Type RM Length L Ch R = 1 ,35500   ,500,500,500
BEGIN DESCRIPTION:
HICKORY CREEK 71.0
END DESCRIPTION:
XS GIS Cut Line= 3
      2755925.77     10210926.25       2756704.1     10210942.61
      2757464.63     10210756.38
#Sta/Elev= 30
  4221.5 1219.64  4421.5 1211.92  4571.5 1199.13  4741.5 1196.25  4786.3 1193.73
  4801.5 1192.53  4831.5 1185.75  4891.6 1181.17  4901.6 1177.19  4911.6 1175.73
  4957.3 1175.06  4958.8 1174.06  5039.2 1175.06  5042.8 1176.45  5094.3 1175.75
  5101.2 1178.47  5125.2 1181.87    5259 1191.43  5314.4 1192.47  5350.9 1195.94
  5403.2  1196.5  5439.3 1200.09    5486 1201.04  5527.6 1203.53  5569.3  1208.4
  5598.8 1208.69  5684.4    1216  5730.6 1223.66  5771.3 1227.67    5783 1229.54
#Mann= 5 ,-1 , 0
  4221.5     .05       0  4957.3     .03       0  5039.2     .05       0
  5684.4     .12       0  5771.3     .05       0
Bank Sta=4957.3,5039.2
XS Rating Curve= 0 ,0
Exp/Cntr=0.3,0.1

Type RM Length L Ch R = 1 ,35000   ,500,500,500
BEGIN DESCRIPTION:
HICKORY CREEK 70.0
END DESCRIPTION:
XS GIS Cut Line= 3
      2755895.83     10211405.88      2756650.05     10211429.57
      2757334.66     10211445.85
#Sta/Elev= 30
  4245.4 1222.81  4415.3 1213.62  4665.5 1197.26  4715.5  1196.5  4775.5 1190.24
  4815.5 1183.64  4895.6 1179.38  4915.6 1176.92  4925.6 1174.01  4944.7 1173.94
  4946.2 1172.94  5025.1 1172.94  5026.6 1173.94  5075.7    1174  5095.7 1179.76
  5105.7 1181.04  5125.7 1180.35  5145.7 1181.32  5165.7 1185.04  5175.7 1184.69
  5191.7 1186.47  5225.7 1188.09  5255.7 1194.78  5290.4 1198.61    5360 1203.07
  5395.7 1206.82  5487.7  1210.9  5575.8 1215.14  5684.2 1217.56  5684.8 1217.56
#Mann= 7 ,-1 , 0
  4245.4     .05       0  4944.7     .03       0  5026.6     .05       0
  5191.7     .12       0  5290.4     .05       0  5487.7     .12       0
  5684.2     .05       0
Bank Sta=4944.7,5026.6
XS Rating Curve= 0 ,0
Exp/Cntr=0.3,0.1

Type RM Length L Ch R = 1 ,34500   ,500,500,500
BEGIN DESCRIPTION:
HICKORY CREEK 69.0
END DESCRIPTION:
XS GIS Cut Line= 3
      2755825.88     10211835.55      2756623.69     10211896.01
      2757309.76     10211925.48
#Sta/Elev= 30
  4199.9 1223.06  4294.1 1216.79  4380.2 1211.13  4420.3 1207.38  4510.6 1201.87
  4580.8 1195.78  4633.4 1193.92    4651 1191.64  4701.1 1188.78  4731.2 1184.93
  4759.7 1183.47  4764.7 1184.26  4801.4 1179.68  4851.6 1179.05  4891.1 1173.87
  4991.1 1172.78  4992.6 1171.78  5071.5 1171.78    5073 1172.78  5082.1 1178.91
  5122.1 1181.16  5279.6 1198.49  5284.6 1197.65  5302.3 1199.76  5422.4 1203.33
  5572.5 1212.74  5602.5 1216.08  5632.6 1217.88  5662.6 1221.61  5686.7 1222.14
#Mann= 4 ,-1 , 0
  4199.9     .12       0  4294.1     .05       0  4991.1     .03       0
    5073     .05       0
Bank Sta=4991.1,5073
XS Rating Curve= 0 ,0
Exp/Cntr=0.3,0.1

Type RM Length L Ch R = 1 ,34000   ,500,500,500
BEGIN DESCRIPTION:
HICKORY CREEK 68.0
END DESCRIPTION:
XS GIS Cut Line= 3
      2755800.92     10211985.45      2756481.17     10212322.78
      2757129.88     10212525.02
#Sta/Elev= 30
  4240.7 1220.93  4338.8 1218.84  4355.6 1215.57  4380.7 1214.13  4488.5 1205.79
  4550.1 1201.52  4579.8 1200.02  4609.8 1196.51  4703.7 1188.72  4764.7 1188.42
  4781.6 1183.99  4809.6 1179.74  4871.1 1177.72  4899.2 1172.34  4972.1 1172.78
  4984.7 1171.57  4986.2 1170.57  5065.1 1170.57  5066.6 1171.57  5084.2  1176.5
    5122 1177.99  5154.5 1181.68  5172.3 1186.27  5219.5 1191.79  5266.6 1195.89
  5354.8 1198.07  5484.8 1212.67  5580.8 1219.82  5620.1 1227.18  5679.5 1230.65
#Mann= 7 ,-1 , 0
  4240.7     .05       0  4380.7     .12       0  4488.5     .05       0
  4550.1     .12       0  4609.8     .05       0  4984.7     .05       0
  5066.6     .05       0
Bank Sta=4984.7,5066.6
XS Rating Curve= 0 ,0
Exp/Cntr=0.3,0.1

Type RM Length L Ch R = 1 ,33500   ,500,500,500
BEGIN DESCRIPTION:
HICKORY CREEK 67.0
END DESCRIPTION:
XS GIS Cut Line= 4
       2755780.9     10212015.38      2755831.42     10212491.83
      2756275.48     10212770.35      2756929.98     10213064.59
#Sta/Elev= 30
  3996.7 1219.33  4064.3 1217.43  4074.5 1217.06  4182.4 1213.15  4306.2 1211.14
  4336.3 1212.16  4366.5 1209.88    4539 1205.49  4764.1 1190.32  4864.3 1177.09
    4894 1175.25  4906.7 1170.95  5005.5 1170.35    5007 1169.35  5085.9 1169.35
  5087.4 1170.35  5098.9 1170.57  5115.9 1175.72  5190.9 1178.54  5274.3 1187.25
  5335.3 1191.04  5363.9 1190.93  5410.3 1194.73  5433.4 1198.85  5462.1 1201.75
  5479.7 1205.43  5485.2 1204.66  5502.9 1207.14  5636.1 1216.26  5717.6 1219.93
#Mann= 5 ,-1 , 0
  3996.7     .05       0  4064.3     .12       0  4074.5     .05       0
  5005.5     .05       0  5087.4     .05       0
Bank Sta=5005.5,5087.4
XS Rating Curve= 0 ,0
Exp/Cntr=0.3,0.1

Type RM Length L Ch R = 1 ,33000   ,500,500,500
BEGIN DESCRIPTION:
HICKORY CREEK 66.0
END DESCRIPTION:
XS GIS Cut Line= 3
      2754486.92     10212694.89      2756061.53     10213206.38
      2756594.15     10213488.68
#Sta/Elev= 30
  3344.4 1220.01  3772.3 1196.33  3841.4 1196.64  3974.5 1187.86  4097.1 1185.99
  4166.3 1180.44  4184.2 1176.01  4278.9 1174.83  4288.8  1177.7  4294.1 1175.74
    4358 1180.75  4373.5 1179.26  4421.9 1184.44  4645.6 1192.64  4688.9 1187.54
  4783.9 1184.15  4906.5 1169.89  4942.4 1168.49  4943.9 1167.49  5024.3 1168.49
  5083.7 1169.09  5095.2 1173.68  5140.5 1175.04  5231.1 1185.52  5287.6 1198.53
    5364 1206.58  5495.9 1214.68  5512.3  1218.2  5539.9 1215.73  5602.8 1217.04
#Mann= 4 ,-1 , 0
  3344.4     .05       0  4942.4     .03       0  5140.5     .05       0
    5364     .05       0
#XS Ineff= 2 , 0
         4628.42 1192.85
Permanent Ineff=
       F       F
Bank Sta=4942.4,5024.3
XS Rating Curve= 0 ,0
Exp/Cntr=0.3,0.1

Type RM Length L Ch R = 1 ,32500   ,500,500,500
BEGIN DESCRIPTION:
HICKORY CREEK 65.0
END DESCRIPTION:
XS GIS Cut Line= 4
      2754901.55     10213269.43      2755446.16     10213524.25
      2755836.34       10213634.      2756389.28     10213848.55
#Sta/Elev= 30
  3993.4 1208.63  4133.9 1203.09  4299.3 1201.71  4339.5 1199.05  4351.3 1199.69
  4406.5 1196.73    4482 1190.46  4561.6 1186.64  4656.5 1183.59  4708.4 1184.28
  4739.6 1182.89  4822.7 1173.98  4834.4 1169.52  4843.5 1168.75    4981 1168.88
  5002.3 1167.79  5003.8 1166.79  5082.8 1166.79  5084.3 1167.79  5085.1 1173.95
  5122.3 1174.25  5170.9 1177.35  5231.2 1189.49  5236.6 1189.19  5261.1 1192.73
  5315.6 1197.75  5417.6 1203.31  5429.9 1202.75  5508.9 1205.38  5593.1 1206.38
#Mann= 4 ,-1 , 0
  3993.4     .05       0  4561.6     .05       0  5002.3     .03       0
  5261.1     .05       0
Bank Sta=5002.3,5084.3
XS Rating Curve= 0 ,0
Exp/Cntr=0.3,0.1

Type RM Length L Ch R = 1 ,32000   ,500,500,500
BEGIN DESCRIPTION:
HICKORY CREEK 64.0
END DESCRIPTION:
XS GIS Cut Line= 4
       2754886.6      10213329.4      2755294.06     10213877.46
      2755588.75     10214064.39      2756400.44     10214113.79
#Sta/Elev= 30
  3968.1 1207.93  4112.5 1200.77  4241.9  1196.1  4477.6 1190.91  4527.6 1191.23
  4533.9 1192.39  4613.2 1190.21  4648.2 1191.63  4655.6 1190.22  4700.7 1190.43
  4722.5 1189.98  4758.6 1186.33  4807.2 1175.98  4843.6 1174.17  4866.1 1168.24
  4931.8 1166.95  4960.8 1167.83    4966 1166.54  4967.5 1165.54  5046.5 1165.54
    5048 1166.54  5147.2 1168.35  5157.2 1171.47  5229.1 1174.27  5258.7 1177.04
  5307.5 1182.52    5430 1191.25  5537.9 1197.28  5678.2 1202.51  5813.2 1204.48
#Mann= 7 ,-1 , 0
  3968.1     .05       0  4700.7     .12       0  4758.6     .05       0
    4966     .05       0    5048     .05       0  5258.7     .12       0
    5430     .05       0
Bank Sta=4966,5048
XS Rating Curve= 0 ,0
Exp/Cntr=0.3,0.1

Type RM Length L Ch R = 1 ,31500   ,500,500,500
BEGIN DESCRIPTION:
HICKORY CREEK 63.0
END DESCRIPTION:
XS GIS Cut Line= 3
      2755081.42     10215232.96      2755538.65     10214550.11
      2756415.39     10214193.74
#Sta/Elev= 30
  4178.2 1211.45  4225.5 1209.17  4303.5 1208.48  4368.7 1204.61  4411.6 1204.06
  4483.7 1199.88  4504.7  1198.2    4533 1193.11  4606.7 1191.22  4663.8 1192.86
  4693.8 1191.98  4750.8 1188.02  4762.9 1185.82  4786.9 1184.49  4874.6 1172.79
    4895 1167.09    4916 1165.27  4954.1 1164.87  4955.6 1163.87  5036.3 1164.87
  5062.7 1166.92  5234.3  1169.4  5266.1 1172.09  5277.5 1171.17  5378.7 1181.34
  5492.6 1188.38  5664.9 1194.57  5753.3 1199.31  5914.3 1204.21  5946.4 1203.98
#Mann= 9 ,-1 , 0
  4178.2     .05       0  4368.7     .12       0    4533     .05       0
  4762.9     .12       0  4874.6     .05       0  4954.1     .03       0
  5036.3     .05       0  5378.7     .12       0  5492.6     .05       0
Bank Sta=4954.1,5036.3
XS Rating Curve= 0 ,0
Exp/Cntr=0.3,0.1

Type RM Length L Ch R = 1 ,31000   ,500,500,500
BEGIN DESCRIPTION:
HICKORY CREEK 62.0
END DESCRIPTION:
XS GIS Cut Line= 3
      2755576.04     10215422.82      2755872.67     10214883.86
      2756455.41     10214238.66
#Sta/Elev= 30
  4384.8 1218.29  4457.7  1211.7  4473.7 1212.43  4517.3 1205.95  4539.1 1205.28
  4555.2 1202.86  4567.1 1198.14  4598.7 1196.12  4620.5  1190.9  4626.2 1191.39
  4642.3 1186.16  4685.9 1181.83  4692.7 1178.42  4707.7 1176.64  4723.7 1176.91
  4751.2 1172.49  4810.9 1172.03  4832.7 1168.66  4886.6 1165.73  4914.1  1167.4
  4932.6 1163.73  4934.1 1162.73  5014.8 1163.73  5108.8 1165.24    5187 1169.12
  5278.7 1179.99    5438 1188.19  5533.7 1190.02  5682.4 1197.47  5869.4 1203.05
#Mann= 5 ,-1 , 0
  4384.8     .05       0  4932.6     .03       0  5014.8     .05       0
  5278.7     .12       0    5438     .05       0
Bank Sta=4932.6,5014.8
XS Rating Curve= 0 ,0
Exp/Cntr=0.3,0.1

Type RM Length L Ch R = 1 ,30500   ,500,500,500
BEGIN DESCRIPTION:
HICKORY CREEK 61.0
END DESCRIPTION:
XS GIS Cut Line= 3
      2755790.86     10215667.62      2756286.01     10215154.45
      2756535.32     10214263.68
#Sta/Elev= 30
  4286.9 1212.66  4321.7 1211.47    4343 1212.49  4420.7 1208.69  4512.8 1201.79
  4533.9 1201.86  4541.1 1200.62  4555.3 1194.96  4562.2 1195.22  4569.4 1192.99
  4654.3 1182.28  4682.3 1180.44  4746.1 1172.81  4837.2 1169.87  4849.2 1169.92
  4901.8 1168.64  4903.1 1162.61  4904.6 1161.61  4983.8 1161.61  4985.3 1162.61
  5022.4 1164.54  5129.9 1164.64  5177.9 1163.04  5242.7 1172.63    5261 1172.81
  5342.3 1178.81  5601.3 1188.25  5670.1 1191.26  5782.2 1196.95    5925 1201.43
#Mann= 9 ,-1 , 0
  4286.9     .05       0  4837.2     .12       0  4849.2     .05       0
  4903.1     .03       0  4985.3     .05       0  5342.3     .12       0
  5601.3     .05       0  5670.1     .12       0  5782.2     .05       0
Bank Sta=4903.1,4985.3
XS Rating Curve= 0 ,0
Exp/Cntr=0.3,0.1

Type RM Length L Ch R = 1 ,30000   ,500,500,500
BEGIN DESCRIPTION:
HICKORY CREEK 60.0
END DESCRIPTION:
XS GIS Cut Line= 3
      2756530.31     10216007.36      2756729.94     10215367.58
      2757029.95     10214713.29
#Sta/Elev= 30
  4329.8 1205.81  4365.2 1204.03  4382.7 1203.53  4418.1 1202.26  4427.5 1199.71
  4432.8 1199.94    4439 1197.86  4464.9 1193.56  4491.4 1192.79    4503 1190.93
  4562.8 1186.79  4600.5 1186.51  4617.1 1183.74  4742.8 1174.46  4889.5 1170.85
  4920.9 1166.78  4921.7 1161.09  4923.2 1160.09  5002.4 1160.09  5003.9 1161.09
  5190.1 1163.43  5213.1 1168.18  5257.9 1171.36    5346 1180.69  5365.9 1181.35
  5558.3  1188.9    5603 1191.04    5610 1192.29  5713.6 1196.34  5719.8 1196.56
#Mann= 9 ,-1 , 0
  4329.8     .12       0  4365.2     .05       0  4382.7     .12       0
  4464.9     .05       0  4921.7     .03       0  5003.9     .05       0
  5365.9     .12       0  5558.3     .05       0  5713.6     .12       0
Bank Sta=4921.7,5003.9
XS Rating Curve= 0 ,0
Exp/Cntr=0.3,0.1

Type RM Length L Ch R = 1 ,29500   ,500,500,500
BEGIN DESCRIPTION:
HICKORY CREEK 59.0
END DESCRIPTION:
XS GIS Cut Line= 3
      2756850.09     10216102.23      2757154.27     10215552.59
      2758212.33      10215163.6
#Sta/Elev= 30
  4371.8 1201.26  4462.2 1198.35  4591.3 1188.53  4640.4 1183.12  4757.8 1174.88
  4862.2 1170.71  4927.9  1165.8  4941.2 1162.96  4955.3  1160.2  5065.4 1160.91
  5171.4 1159.77  5172.9 1158.77  5252.3 1158.77  5253.8 1159.77  5257.2 1161.08
  5298.6 1161.17  5329.1 1166.35  5359.6 1166.77  5429.7 1174.18  5470.3 1177.13
  5576.8 1176.72  5684.1 1179.22  5825.8 1186.34  5842.1 1188.55  5860.2 1192.08
    5869 1192.87  5911.9 1197.94  5937.1 1202.33  5981.7 1205.92  6127.3    1209
#Mann= 10 ,-1 , 0
  4371.8     .12       0  4591.3     .05       0  4757.8     .12       0
  4941.2     .05       0  5171.4     .03       0  5253.8     .05       0
  5429.7     .12       0  5842.1     .05       0  5860.2     .12       0
    5869     .05       0
Bank Sta=5171.4,5253.8
XS Rating Curve= 0 ,0
Exp/Cntr=0.3,0.1

Type RM Length L Ch R = 1 ,29000   ,500,500,500
BEGIN DESCRIPTION:
HICKORY CREEK 58.0
END DESCRIPTION:
XS GIS Cut Line= 3
      2756954.96     10216252.16        2757585.     10215758.35
      2758098.71     10215507.91
#Sta/Elev= 30
  4199.5 1197.36  4294.2 1194.63  4441.8 1188.53  4469.5 1185.55    4567 1180.53
  4589.1  1179.5    4738 1170.41  4770.6 1168.96  4848.3 1168.69  4911.9 1163.21
  4925.2 1159.12  4970.7 1158.41  4972.2 1157.41  5051.6 1157.41  5053.1 1158.41
  5167.6 1159.56  5178.1  1160.8  5189.9 1164.73  5228.8 1168.65  5256.9 1174.27
  5288.1 1178.14  5341.5 1183.75    5347 1185.93  5356.8 1185.92  5414.6 1197.68
  5423.5 1197.83  5459.7 1204.28  5499.2 1203.95  5550.1 1208.75  5571.5 1210.14
#Mann= 10 ,-1 , 0
  4199.5     .12       0  4294.2     .05       0    4567     .12       0
  4589.1     .05       0    4738     .12       0  4770.6     .05       0
  4970.7     .03       0  5053.1     .05       0  5288.1     .12       0
  5550.1     .05       0
Bank Sta=4970.7,5053.1
XS Rating Curve= 0 ,0
Exp/Cntr=0.3,0.1

Type RM Length L Ch R = 1 ,28500   ,500,500,500
BEGIN DESCRIPTION:
HICKORY CREEK 57.0
END DESCRIPTION:
XS GIS Cut Line= 3
      2756890.08     10216362.05      2757826.78     10216189.85
      2758512.25     10216406.53
#Sta/Elev= 30
  4047.6 1197.64  4155.5  1193.1  4358.3 1187.67  4384.6 1185.77  4449.8 1182.51
  4482.4 1182.48  4551.5 1182.17  4561.7 1180.09  4658.3 1174.86  4736.3  1168.8
  4784.3 1162.89  4789.4 1163.72  4795.5 1161.14  4805.7 1160.02  4978.6 1156.71
  4980.1 1155.71    5061 1156.71  5063.8 1162.55  5109.6  1167.5  5145.7 1174.11
  5198.3 1177.25  5250.6 1177.69  5299.1 1181.74  5354.7 1184.22  5392.3 1189.16
  5431.6 1189.31  5469.2 1190.73  5586.2 1191.04  5656.1 1196.98  5718.9 1199.29
#Mann= 11 ,-1 , 0
  4047.6     .05       0  4155.5     .12       0  4384.6     .05       0
  4482.4     .12       0  4658.3     .05       0  4978.6     .05       0
    5061     .05       0  5109.6     .12       0  5299.1     .05       0
  5431.6     .12       0  5469.2     .05       0
Bank Sta=4978.6,5061
XS Rating Curve= 0 ,0
Exp/Cntr=0.3,0.1

Type RM Length L Ch R = 1 ,28000   ,500,500,500
BEGIN DESCRIPTION:
HICKORY CREEK 56.0
END DESCRIPTION:
XS GIS Cut Line= 4
      2756780.13     10216417.01      2757354.68     10216347.07
      2757595.25     10216596.87      2758005.69     10217003.12
#Sta/Elev= 30
  4074.4 1198.12  4130.4 1198.36  4262.7 1193.65  4481.8  1185.3  4583.7 1178.77
  4641.8 1180.33  4693.5 1178.74  4785.6 1171.26  4813.9 1166.65  4842.1 1159.64
  4949.4 1155.46  4950.9 1154.46  5031.8 1155.46    5033 1157.79  5047.1 1159.46
  5075.4 1160.76  5082.5 1158.54  5089.6 1161.33    5132 1162.14  5167.4  1165.9
  5188.6    1165  5287.6 1172.98  5301.7 1175.07  5337.1 1184.69  5344.1 1184.05
  5379.4 1189.19    5429 1193.44  5457.3 1193.56  5492.7 1198.72  5577.5 1206.92
#Mann= 6 ,-1 , 0
  4074.4     .05       0  4262.7     .12       0  4481.8     .05       0
  4949.4     .05       0  5031.8     .05       0  5379.4     .12       0
Bank Sta=4949.4,5031.8
XS Rating Curve= 0 ,0
Exp/Cntr=0.3,0.1

Type RM Length L Ch R = 1 ,27500   ,500,500,500
BEGIN DESCRIPTION:
HICKORY CREEK 55.0
END DESCRIPTION:
XS GIS Cut Line= 3
      2756760.17     10216536.94       2757249.7     10216940.76
      2757869.27     10217356.28
#Sta/Elev= 30
  4365.4 1192.47  4427.6 1190.36    4523  1189.2  4615.5  1185.5    4665 1181.97
  4728.9 1173.23  4771.9 1176.95  4786.2 1175.62  4813.5 1168.03  4827.9 1166.19
  4864.4 1165.93  4878.1 1168.29  4899.6 1167.12  4928.2 1159.99  4928.7 1154.09
  4930.2 1153.09  5011.1 1154.09  5157.3 1156.22  5172.3 1159.15  5301.3 1165.75
  5344.3 1170.83  5409.4 1172.89  5496.4 1178.96  5589.4 1188.63  5619.4  1188.8
  5661.5 1192.95  5676.5  1191.5    5701 1192.96  5744.1  1194.8    5746  1194.8
#Mann= 6 ,-1 , 0
  4365.4     .12       0  4427.6     .05       0  4928.7     .03       0
  5011.1     .05       0    5701     .12       0  5744.1     .05       0
Bank Sta=4928.7,5011.1
XS Rating Curve= 0 ,0
Exp/Cntr=0.3,0.1

Type RM Length L Ch R = 1 ,27000   ,500,500,500
BEGIN DESCRIPTION:
HICKORY CREEK 54.0
END DESCRIPTION:
XS GIS Cut Line= 3
       2756260.5      10216936.6      2757135.58     10217411.62
      2757772.55     10217660.34
#Sta/Elev= 30
  4004.3 1201.34  4004.9 1201.24  4049.7  1196.9  4065.9 1197.85  4093.4 1195.98
  4143.4 1195.86  4262.6 1192.67  4300.6 1193.91  4306.3 1192.88  4431.8 1192.91
  4595.3 1182.11  4758.8 1175.65  4889.9 1161.63  4911.8 1157.28  4920.5 1153.71
  4933.6 1154.05  4936.2 1152.85  4937.7 1151.85  5018.6 1152.85  5053.8 1154.07
  5095.8 1153.33  5107.5  1157.4  5125.7 1159.78  5185.4 1162.88    5249 1168.76
  5348.4 1174.92  5396.8 1180.65  5541.2  1191.8  5602.9 1198.07  5683.8 1206.93
#Mann= 8 ,-1 , 0
  4004.3     .05       0  4004.9     .12       0  4143.4     .05       0
  4936.2     .05       0  5018.6     .05       0    5249     .12       0
  5396.8     .05       0  5602.9     .12       0
Bank Sta=4936.2,5018.6
XS Rating Curve= 0 ,0
Exp/Cntr=0.3,0.1

Type RM Length L Ch R = 1 ,26500   ,500,500,500
BEGIN DESCRIPTION:
HICKORY CREEK 53.0
END DESCRIPTION:
XS GIS Cut Line= 3
      2756210.55     10218325.55      2757010.31     10217872.84
      2757849.34     10217775.96
#Sta/Elev= 30
    4081 1201.53  4155.3 1197.65  4364.2  1186.7  4600.9 1179.73  4687.5 1178.78
  4768.3 1173.23  4805.8 1168.13  4811.6 1168.77  4833.8 1166.65  4843.4  1163.7
    4865 1161.22  4908.3 1160.03  4910.3 1151.41  4911.8 1150.41  4991.4 1150.41
  4992.9 1151.41  4994.6 1152.39  5146.3 1153.11  5176.5 1159.71  5206.7 1160.45
  5245.2 1164.18  5337.6 1171.59  5377.9 1177.11  5391.4 1176.83    5453 1181.16
  5538.9 1186.35  5639.6 1194.56  5760.5 1200.79  5780.5 1202.08  5844.6 1201.79
#Mann= 7 ,-1 , 0
    4081     .12       0  4155.3     .05       0  4910.3     .03       0
  4992.9     .05       0  5245.2     .12       0    5453     .05       0
  5760.5     .12       0
Bank Sta=4910.3,4992.9
XS Rating Curve= 0 ,0
Exp/Cntr=0.3,0.1

Type RM Length L Ch R = 1 ,26000   ,500,500,500
BEGIN DESCRIPTION:
HICKORY CREEK 52.0
END DESCRIPTION:
XS GIS Cut Line= 3
      2756200.59     10218805.16      2757098.22     10218352.96
      2757909.24     10217885.89
#Sta/Elev= 30
  3994.9 1192.39  4080.9 1197.69  4147.8 1199.22  4214.7 1198.59    4371 1193.17
  4460.2 1186.47  4560.5  1182.3  4594.1 1178.39  4610.8 1179.09  4638.8 1176.14
  4811.6 1167.97  4900.8 1159.85  4904.1 1150.15  4905.6 1149.15  4986.7 1150.15
  5204.6 1153.75  5239.4 1163.89    5285 1167.26  5320.2 1173.04  5516.8 1178.89
  5591.1 1183.52  5650.8 1184.78  5767.8 1186.44  5826.7 1188.17  5832.5 1189.52
  5848.3 1188.02  5885.6 1188.65  5897.2 1190.27  5920.3 1188.33  5935.9 1189.17
#Mann= 6 ,-1 , 0
  3994.9     .12       0  4214.7     .05       0  4904.1     .03       0
  4986.7     .05       0  5516.8     .12       0  5650.8     .05       0
Bank Sta=4904.1,4986.7
XS Rating Curve= 0 ,0
Exp/Cntr=0.3,0.1

Type RM Length L Ch R = 1 ,25500   ,500,500,500
BEGIN DESCRIPTION:
HICKORY CREEK 51.0
END DESCRIPTION:
XS GIS Cut Line= 3
      2757299.72     10219369.74      2757415.39     10218694.48
      2758033.13     10218016.91
#Sta/Elev= 30
  4314.9 1193.17  4585.4 1180.22  4721.5 1169.34  4757.9  1167.8    4799 1161.93
  4879.6 1157.68  4930.4  1149.6  4966.9 1148.52  4968.4 1147.52  5049.5 1148.52
  5050.8 1150.25  5085.9 1150.84  5100.1 1152.59  5199.4 1154.33  5213.6  1157.6
  5248.8 1157.92  5270.4 1160.81  5284.6 1160.31  5291.3 1157.42  5319.7 1162.85
  5354.8 1166.74  5397.3 1168.92  5447.4  1172.6  5496.7  1170.2  5557.4 1174.45
  5673.7 1184.45    5769 1187.28  5864.9 1191.19  5907.5 1194.16  5916.9 1196.59
#Mann= 7 ,-1 , 0
  4314.9     .12       0  4721.5     .05       0  4966.9     .03       0
  5049.5     .05       0  5397.3     .12       0  5557.4     .05       0
    5769     .12       0
Bank Sta=4966.9,5049.5
XS Rating Curve= 0 ,0
Exp/Cntr=0.3,0.1

Type RM Length L Ch R = 1 ,25000   ,500,500,500
BEGIN DESCRIPTION:
HICKORY CREEK 50.0
END DESCRIPTION:
XS GIS Cut Line= 3
      2757744.39     10219374.69      2757880.92     10218824.16
      2758174.04     10218180.68
#Sta/Elev= 30
  4432.8 1193.96  4506.5 1188.77  4609.6 1184.32  4630.2 1181.95  4661.1 1181.21
  4666.5 1182.27  4702.3 1175.94  4707.8 1173.77  4743.5  1172.5  4784.7 1164.13
  4856.8 1157.84  4949.6 1153.54  4956.1 1152.15  4958.2 1146.99  4959.7 1145.99
  5040.8 1146.99  5043.6 1148.35  5187.4 1149.24  5231.9 1150.94  5290.6 1159.43
  5319.8 1168.31  5359.8 1169.66  5382.8 1174.24  5404.7 1176.39  5426.4 1177.47
  5473.7  1178.8  5509.1 1183.04  5555.2 1184.13  5616.5 1188.15  5707.1 1190.42
#Mann= 5 ,-1 , 0
  4432.8     .05       0  4958.2     .03       0  5040.8     .05       0
  5404.7     .12       0  5426.4     .05       0
Bank Sta=4958.2,5040.8
XS Rating Curve= 0 ,0
Exp/Cntr=0.3,0.1

Type RM Length L Ch R = 1 ,24500   ,500,500,500
BEGIN DESCRIPTION:
HICKORY CREEK 49.0
END DESCRIPTION:
XS GIS Cut Line= 3
      2758303.96     10219334.73      2758376.49     10218810.62
      2758455.69     10218303.06
#Sta/Elev= 30
  4470.9 1188.67  4610.1 1178.33  4667.6 1175.99  4739.4 1170.67  4807.3 1163.09
  4825.9 1162.25  4876.3 1155.47  4883.1 1155.24  4888.1 1157.36  4905.9 1152.24
  4916.7 1152.64  4925.9 1145.36  4927.4 1144.36    5007 1144.36  5008.5 1145.36
  5048.1 1151.29  5068.3 1147.67  5108.8 1148.63  5218.4 1146.14  5286.3 1161.94
  5300.9 1162.98  5321.4  1168.5  5354.1 1170.76  5361.8 1173.73    5372  1175.2
  5440.2 1179.71  5452.9 1181.07  5479.7 1186.97  5484.8 1186.63  5513.7 1191.42
#Mann= 8 ,-1 , 0
  4470.9     .12       0  4610.1     .05       0  4807.3     .12       0
  4905.9     .05       0  4925.9     .05       0  5008.5     .05       0
  5300.9     .12       0  5440.2     .05       0
Bank Sta=4925.9,5008.5
XS Rating Curve= 0 ,0
Exp/Cntr=0.3,0.1

Type RM Length L Ch R = 1 ,24000   ,500,500,500
BEGIN DESCRIPTION:
HICKORY CREEK 48.0
END DESCRIPTION:
XS GIS Cut Line= 3
      2758955.69     10219103.13      2758862.29     10218710.79
      2758505.69     10218203.12
#Sta/Elev= 30
  4596.7 1183.52  4624.7 1180.41  4720.1 1173.45  4746.8 1169.19  4751.9 1170.15
  4777.1 1167.26    4789 1165.61  4802.3 1166.19  4836.2 1159.29  4853.7 1153.64
  4879.2 1151.82  4884.5 1150.88  4894.6 1144.31  4896.1 1143.31  4977.3 1144.31
  4987.3 1145.53    5000 1144.35  5160.8 1146.12  5217.4 1155.94  5276.6 1156.25
  5297.6 1158.91  5303.7 1157.58  5327.1  1159.6  5348.1 1163.24    5369 1164.47
  5419.6 1175.52  5449.2 1175.92  5526.7 1186.86  5583.7 1197.79  5620.4 1201.93
#Mann= 6 ,-1 , 0
  4596.7     .12       0  4624.7     .05       0  4777.1     .12       0
  4879.2     .05       0  4894.6     .05       0  4977.3     .05       0
Bank Sta=4894.6,4977.3
XS Rating Curve= 0 ,0
Exp/Cntr=0.3,0.1

Type RM Length L Ch R = 1 ,23500   ,500,500,500
BEGIN DESCRIPTION:
HICKORY CREEK 47.0
END DESCRIPTION:
XS GIS Cut Line= 3
      2759363.13     10219094.98      2759356.76     10218678.93
       2759238.4     10217887.02
#Sta/Elev= 30
  4583.9 1181.17  4715.8 1173.19  4805.8 1169.86  4817.2 1168.33  4885.8 1161.03
  4915.8 1153.28  4935.8 1150.89  4955.8 1149.75  4964.5 1143.14    4966 1142.14
  5045.7 1142.14  5047.2 1143.14  5137.3 1143.61    5198 1146.86  5228.3 1145.77
  5265.5 1150.19  5278.9  1150.7  5299.1 1148.25    5313 1148.22  5339.5 1153.96
  5382.2 1157.66  5410.3 1162.82  5460.9  1164.9  5608.4 1176.16  5642.9 1179.05
  5648.9 1180.34  5718.2 1183.36    5744 1186.45  5753.4 1186.75  5800.7 1189.13
#Mann= 7 ,-1 , 0
  4583.9     .12       0  4817.2     .05       0  4964.5     .03       0
  5047.2     .05       0  5265.5     .12       0  5608.4     .05       0
  5753.4     .12       0
Bank Sta=4964.5,5047.2
XS Rating Curve= 0 ,0
Exp/Cntr=0.3,0.1

Type RM Length L Ch R = 1 ,23000   ,500,500,500
BEGIN DESCRIPTION:
HICKORY CREEK 46.0
END DESCRIPTION:
XS GIS Cut Line= 3
      2759747.83     10219279.77      2759697.74     10218464.71
      2759805.69     10217953.07
#Sta/Elev= 30
  4183.4 1177.46  4330.3 1171.61  4360.4 1173.28  4450.6  1169.1  4470.6 1166.89
  4580.8 1164.12  4625.9 1162.46  4640.9  1160.8    4661 1161.05    4681 1157.56
  4811.2 1143.66  4921.4 1139.33  4954.2 1139.99  4956.9 1138.55  4958.4 1137.55
  5038.1 1137.55  5039.6 1138.55  5042.5 1141.63  5083.4 1144.46  5110.1 1147.61
  5115.2 1145.36  5134.5 1148.88  5159.8 1149.18  5216.3 1155.47  5259.4 1157.65
  5277.6  1160.6    5298 1166.15  5318.5  1165.7  5369.6 1168.54  5522.9  1181.5
#Mann= 3 ,-1 , 0
  4183.4     .05       0  4956.9     .05       0  5039.6     .05       0
Bank Sta=4956.9,5039.6
XS Rating Curve= 0 ,0
Exp/Cntr=0.3,0.1

Type RM Length L Ch R = 1 ,22500   ,500,500,500
BEGIN DESCRIPTION:
HICKORY CREEK 45.0
END DESCRIPTION:
XS GIS Cut Line= 3
      2760252.44     10219269.76      2760172.59     10218520.61
      2760277.42     10218070.76
#Sta/Elev= 30
  4246.6  1174.1  4424.3 1170.14    4555 1162.39  4605.3    1163  4645.6 1158.98
  4695.8 1159.74    4726 1155.64  4830.4 1150.25    4907 1140.57  4976.6 1137.73
  4978.1 1136.73  5057.8 1136.73  5059.3 1137.73  5077.1 1138.87  5124.8 1138.41
  5130.9 1141.56  5151.4 1146.19  5215.2 1148.52  5243.9 1157.24  5252.5 1162.67
  5257.6 1162.27  5274.7 1172.87  5284.9 1176.47  5295.1 1177.95  5300.2 1176.96
    5326 1178.51  5347.9  1177.9  5358.8 1179.33  5397.9 1186.37  5461.9 1188.17
#Mann= 5 ,-1 , 0
  4246.6     .05       0  4976.6     .03       0  5059.3     .05       0
  5215.2     .12       0  5358.8     .05       0
Bank Sta=4976.6,5059.3
XS Rating Curve= 0 ,0
Exp/Cntr=0.3,0.1

Type RM Length L Ch R = 1 ,22000   ,500,500,500
BEGIN DESCRIPTION:
HICKORY CREEK 44.0
END DESCRIPTION:
XS GIS Cut Line= 4
      2760457.28     10219289.81      2760659.82     10218563.62
      2760610.82     10218237.31      2760478.14     10218056.92
#Sta/Elev= 30
  4246.1 1171.94    4388 1170.61  4585.3 1164.68  4699.5 1159.75  4730.6  1156.2
  4750.8 1155.22    4824 1148.15  4881.4 1145.26  4917.5 1143.77  4925.7 1142.05
    4959 1139.75  4969.3  1136.8  4970.8  1135.8  5050.5  1135.8    5052  1136.8
  5162.3 1137.07  5172.4 1139.06  5182.5 1143.67    5223 1148.84  5252.8 1155.65
    5266 1160.36  5303.9 1162.04  5328.5 1165.02  5372.4 1174.49  5394.4 1176.41
  5436.1 1177.63  5486.2 1181.35  5515.5 1181.15  5521.7 1182.17  5553.9 1182.86
#Mann= 7 ,-1 , 0
  4246.1     .05       0  4750.8     .12       0  4881.4     .05       0
  4969.3     .03       0    5052     .05       0  5252.8     .12       0
  5328.5     .05       0
Bank Sta=4969.3,5052
XS Rating Curve= 0 ,0
Exp/Cntr=0.3,0.1

Type RM Length L Ch R = 1 ,21500   ,500,500,500
BEGIN DESCRIPTION:
HICKORY CREEK 43.0
END DESCRIPTION:
XS GIS Cut Line= 3
      2760542.22     10219274.81      2761129.02     10218647.88
      2761570.22     10218027.47
#Sta/Elev= 30
  4141.3 1169.87  4237.1 1168.47  4314.7 1169.68  4455.1 1161.81  4725.7 1147.54
  4795.9 1143.33  4845.2 1142.38  4866.7 1138.49  4880.9  1137.1  5031.2  1135.3
  5032.7  1134.3  5112.5  1134.3    5114  1135.3  5116.3 1142.25  5137.9 1144.64
  5158.7 1146.24  5202.2 1154.51  5223.9 1155.63    5230 1156.92  5280.5 1158.53
  5379.3 1165.43  5486.2 1170.07    5503 1171.52  5508.3 1171.08  5538.7 1171.57
  5660.5 1176.86  5710.9  1179.9  5722.9 1182.32  5746.5 1182.16  5761.3 1183.61
#Mann= 10 ,-1 , 0
  4141.3     .05       0  4455.1     .12       0  4725.7     .05       0
  5031.2     .03       0    5114     .05       0  5137.9     .12       0
  5379.3     .05       0  5486.2     .12       0  5508.3     .05       0
  5722.9     .12       0
Bank Sta=5031.2,5114
XS Rating Curve= 0 ,0
Exp/Cntr=0.3,0.1

Type RM Length L Ch R = 1 ,21000   ,500,500,500
BEGIN DESCRIPTION:
HICKORY CREEK 42.0
END DESCRIPTION:
XS GIS Cut Line= 3
      2760542.18     10219329.78      2761450.78      10219012.2
      2761990.88       10219015.
#Sta/Elev= 30
  4037.5 1169.66    4126 1167.64  4231.9 1168.08  4337.8 1166.15    4412  1161.4
  4592.7  1154.3  4649.5 1149.87  4655.6 1148.67  4773.7 1141.96  4799.4 1138.54
  4830.5 1136.67  4892.6 1135.75  4918.3 1134.29  4999.9 1134.22  5003.5  1133.2
    5005  1132.2  5084.8  1132.2  5086.3  1133.2  5094.9 1143.63  5104.9 1144.15
  5154.9  1150.6    5196 1153.27  5244.9 1155.08  5274.9 1161.67  5294.8 1163.31
  5393.5 1167.93  5424.9 1169.38  5454.9 1172.31  5474.9 1171.83  5540.1 1173.63
#Mann= 6 ,-1 , 0
  4037.5     .05       0  5003.5     .03       0  5086.3     .05       0
    5196     .12       0  5294.8     .05       0  5393.5     .12       0
Bank Sta=5003.5,5086.3
XS Rating Curve= 0 ,0
Exp/Cntr=0.3,0.1

Type RM Length L Ch R = 1 ,20500   ,500,500,500
BEGIN DESCRIPTION:
HICKORY CREEK 41.0
END DESCRIPTION:
XS GIS Cut Line= 3
      2760527.28     10219389.72      2761290.25     10219444.02
      2761930.92     10219549.55
#Sta/Elev= 30
  4235.1 1168.83  4383.9 1163.93  4491.7 1165.55  4604.4 1163.63  4734.8 1151.94
  4804.9 1146.92  4855.1 1141.29  4885.1 1133.46  4945.3 1133.49  4986.6 1131.11
  4988.1 1130.11  5067.9 1130.11  5069.4 1131.11  5076.5 1132.51  5096.7 1131.81
  5150.3 1133.63  5206.4 1142.21  5272.7 1147.28  5350.1 1155.31  5360.2 1154.35
  5370.4 1155.03  5380.5 1153.51  5389.9 1155.93    5395 1155.14  5400.8 1157.01
  5410.9 1157.92  5456.2 1159.92  5481.8 1162.43  5578.5  1167.2  5649.3 1168.82
#Mann= 3 ,-1 , 0
  4235.1     .05       0  4986.6     .03       0  5069.4     .05       0
Bank Sta=4986.6,5069.4
XS Rating Curve= 0 ,0
Exp/Cntr=0.3,0.1

Type RM Length L Ch R = 1 ,20000   ,500,500,500
BEGIN DESCRIPTION:
HICKORY CREEK 40.0
END DESCRIPTION:
XS GIS Cut Line= 3
      2760197.44     10219769.42      2761101.65     10219886.01
       2761896.2     10219984.26
#Sta/Elev= 30
  4088.3 1183.99  4122.3 1181.43  4207.5 1177.12  4288.2 1169.63  4520.1 1155.61
  4546.3 1152.29  4610.8 1153.73  4728.8 1152.97  4772.2 1152.17  4836.3  1141.2
  4842.7  1140.2  4858.9 1133.72    4873 1131.77  4992.9 1129.88  4994.4 1128.88
  5075.7 1129.88  5084.7 1133.16  5180.2 1134.99  5185.4 1137.48  5195.5 1137.96
  5215.4 1137.09  5225.7 1137.09  5245.9 1140.92  5274.8 1141.07  5296.3 1143.26
  5428.4 1147.98  5607.3 1158.85  5679.2 1164.06  5770.8 1167.15  5800.6 1167.82
#Mann= 10 ,-1 , 0
  4088.3     .12       0  4122.3     .05       0  4728.8     .12       0
  4836.3     .05       0  4992.9     .05       0  5075.7     .05       0
  5215.4     .12       0  5274.8     .05       0  5607.3     .12       0
  5770.8     .05       0
Bank Sta=4992.9,5075.7
XS Rating Curve= 0 ,0
Exp/Cntr=0.3,0.1

Type RM Length L Ch R = 1 ,19500   ,500,500,500
BEGIN DESCRIPTION:
HICKORY CREEK 39.0
END DESCRIPTION:
XS GIS Cut Line= 3
      2760337.39     10220373.96      2760924.63     10220310.15
      2761936.15     10220169.11
#Sta/Elev= 30
  4409.3  1182.2  4651.3 1169.86  4799.8 1159.13  4834.4 1155.65  4890.4 1147.69
  4920.6 1140.05    4926 1136.41    4931 1137.04  4940.7 1133.58  4949.6 1128.54
  4951.1 1127.54  5030.9 1127.54  5032.4 1128.54  5051.5  1128.9  5061.6 1130.43
  5092.1 1129.33  5132.3 1130.02  5152.5 1132.62  5235.2 1137.51  5263.6 1137.82
  5292.7 1135.96  5306.7 1135.87  5384.7 1144.69  5463.6 1145.01    5516 1143.28
    5576 1145.47  5643.9  1148.8    5823 1158.81  5937.4 1164.75  6021.3 1166.23
#Mann= 10 ,-1 , 0
  4409.3     .05       0  4799.8     .12       0  4949.6     .03       0
  5032.4     .12       0  5292.7     .12       0  5463.6     .05       0
    5576     .12       0  5643.9     .05       0    5823     .12       0
  5937.4     .05       0
Bank Sta=4949.6,5032.4
XS Rating Curve= 0 ,0
Exp/Cntr=0.3,0.1

Type RM Length L Ch R = 1 ,19000   ,500,500,500
BEGIN DESCRIPTION:
HICKORY CREEK 38.0
END DESCRIPTION:
XS GIS Cut Line= 3
      2760467.31     10220903.54      2761037.34     10220783.19
       2762080.9     10220523.87
#Sta/Elev= 30
  4417.4 1169.62    4542 1164.68  4650.8 1157.82  4691.7 1152.32  4780.6  1147.8
  4785.7 1148.64  4793.9 1146.78  4824.6 1145.04  4880.1 1139.22  4906.3  1134.7
  4947.2 1131.08  4967.1 1127.74  4968.6 1126.74  5048.5 1126.74    5050 1127.74
  5132.2 1130.74  5194.1 1130.56  5286.8 1141.58  5348.9 1143.87  5410.5 1142.63
  5464.5 1144.19  5554.7 1146.52  5657.5 1149.29  5676.8 1150.01  5740.2 1152.81
  5760.4 1155.26  5895.9 1158.31  5905.1 1157.27  5915.4 1158.85  6075.3 1165.86
#Mann= 9 ,-1 , 0
  4417.4     .05       0  4967.1     .03       0    5050     .05       0
  5348.9     .12       0  5464.5     .05       0  5554.7     .12       0
  5657.5     .05       0  5676.8     .12       0  5760.4     .05       0
Bank Sta=4967.1,5050
XS Rating Curve= 0 ,0
Exp/Cntr=0.3,0.1

Type RM Length L Ch R = 1 ,18500   ,500,500,500
BEGIN DESCRIPTION:
HICKORY CREEK 37.0
END DESCRIPTION:
XS GIS Cut Line= 3
      2760502.24     10221613.01      2761314.29      10221178.5
      2762056.04     10220888.56
#Sta/Elev= 30
    4079 1174.45  4083.8 1174.45    4089 1171.54  4116.9  1168.1  4149.1 1165.63
  4207.7 1164.34  4287.1 1156.42  4406.7  1154.4  4592.8 1145.11  4620.5 1146.38
  4658.7 1144.46  4686.3 1148.23  4708.2 1148.19  4842.8 1139.47    4900 1129.33
  4992.3 1126.48  4993.8 1125.48  5075.2 1126.48  5076.6 1129.25  5082.7 1129.55
  5191.4 1129.13    5227 1136.46  5259.2 1140.29  5368.2 1144.72    5476 1148.36
  5559.8 1154.77  5613.5 1155.45  5645.7 1158.29  5661.1 1157.46  5796.4 1162.92
#Mann= 5 ,-1 , 0
    4079     .05       0  4992.3     .03       0  5075.2     .05       0
  5368.2     .12       0    5476     .05       0
Bank Sta=4992.3,5075.2
XS Rating Curve= 0 ,0
Exp/Cntr=0.3,0.1

Type RM Length L Ch R = 1 ,18000   ,500,500,500
BEGIN DESCRIPTION:
HICKORY CREEK 36.0
END DESCRIPTION:
XS GIS Cut Line= 3
      2760866.98     10221877.79      2761481.91     10221626.75
      2762150.82     10221278.34
#Sta/Elev= 30
  4335.8 1159.57  4516.4 1150.58  4582.8 1150.37  4599.3 1149.05  4628.7 1149.98
  4647.3 1148.15  4652.7 1148.81  4658.4 1147.09  4682.2 1146.97  4730.2 1142.71
  4813.1 1139.11  4938.7 1126.56  4982.5 1126.69  5014.3 1125.29  5026.8  1127.8
    5042 1129.01  5058.5 1125.41  5094.5 1127.72  5102.7 1126.62  5174.6 1126.51
  5177.4 1124.54  5178.9 1123.54  5258.8 1123.54  5260.3 1124.54  5286.1 1127.96
  5295.9 1132.04  5340.1  1139.6  5400.8 1143.92  5514.8 1149.46  5754.2 1158.17
#Mann= 5 ,-1 , 0
  4335.8     .05       0  5177.4     .03       0  5260.3     .05       0
  5400.8     .12       0  5514.8     .05       0
Bank Sta=5177.4,5260.3
XS Rating Curve= 0 ,0
Exp/Cntr=0.3,0.1

Type RM Length L Ch R = 1 ,17500   ,500,500,500
BEGIN DESCRIPTION:
HICKORY CREEK 35.0
END DESCRIPTION:
XS GIS Cut Line= 3
      2760936.92     10222197.55      2761584.01     10222064.62
      2762335.85     10221573.02
#Sta/Elev= 30
  4339.4 1156.41  4435.6 1152.51  4485.9 1153.24  4631.9  1145.9  4682.3 1141.41
  4737.8 1142.72  4766.9 1139.61  4797.5  1141.7  4833.4 1137.87  4848.6 1139.06
  4883.8 1137.58  4929.1 1133.05  4934.2 1134.03    4938 1122.68  4939.5 1121.68
  5020.9 1122.68  5145.6 1125.51  5169.3 1129.55  5205.1 1131.76    5212  1127.7
  5248.2 1123.82  5305.5 1129.51  5320.6 1133.03  5326.6 1132.17  5388.1 1137.22
  5450.2 1141.32  5507.5 1141.91  5667.4 1150.27  5764.1  1153.3  5898.3 1157.73
#Mann= 5 ,-1 , 0
  4339.4     .05       0    4938     .03       0  5020.9     .05       0
  5388.1     .12       0  5764.1     .05       0
Bank Sta=4938,5020.9
XS Rating Curve= 0 ,0
Exp/Cntr=0.3,0.1
