--- LEFT HAND CREEK.prj (project) ---

Proj Title=LEFT HAND CREEK Base Level Engineering
Current Plan=p01
Default Exp/Contr=0.3,0.1
English Units
Geom File=g01
Flow File=f01
Plan File=p01
BEGIN DESCRIPTION:
LEFT HAND CREEK
END DESCRIPTION:

--- LEFT HAND CREEK.p01 (plan) ---

Plan Title=Multiple Run
Short Identifier=Multiple
Geom File=g01
Flow File=f01
Subcritical Flow
K Sum by GR= 0
Std Step Tol= 0.01
Critical Tol= 0.01
Num of Std Step Trials= 20
Max Error Tol= 0.3
Flow Tol Ratio= 0.001
Split Flow NTrial= 30
Split Flow Tol= 0.02
Split Flow Ratio= 0.02
Log Output Level= 0
Friction Slope Method= 1
Unsteady Friction Slope Method= 2
Unsteady Bridges Friction Slope Method= 1
Parabolic Critical Depth
Global Vel Dist=  1 , 1 , 1
Global Log Level= 0
CheckData=True
Encroach Param= -1, 0, 0, 0
BEGIN DESCRIPTION:
Multiple Run
END DESCRIPTION:

--- LEFT HAND CREEK.f01 (steady flow) ---

Flow Title=Multiple
Number of Profiles=7
Profile Names=10-year,25-year,50-year,1pct_min,100-year,1pct_plu,500-year
River Rch & RM= LEFT HAND CREEK,Reach-1,34000
     489     800    1288     965    1766    3233    2495
River Rch & RM= LEFT HAND CREEK,Reach-1,25500
     703    1179    1871    1352    2588    4955    3635
River Rch & RM= LEFT HAND CREEK,Reach-1,21000
     842    1427    2301    1651    3204    6215    4491
River Rch & RM= LEFT HAND CREEK,Reach-1,19000
     992    1693    2862    2082    4013    7734    5614
River Rch & RM= LEFT HAND CREEK,Reach-1,18500
    1067    1832    3053    2188    4287    8400    5994
River Rch & RM= LEFT HAND CREEK,Reach-1,16500
    1354    2353    4085    2951    5786   11341    8057
River Rch & RM= LEFT HAND CREEK,Reach-1,14500
    1532    2691    4746    3370    6771   13605    9467
River Rch & RM= LEFT HAND CREEK,Reach-1,10500
    1638    2888    5129    3628    7337   14838   10258
River Rch & RM= LEFT HAND CREEK,Reach-1,9000
    1853    3297    5880    4115    8451   17355   11815
River Rch & RM= LEFT HAND CREEK,Reach-1,5500
    1886    3361    5946    4140    8544   17633   11940
River Rch & RM= LEFT HAND CREEK,Reach-1,5000
    2254    4066    7149    4911   10317   21674   14374
Boundary for River Rch & Prof#=LEFT HAND CREEK,Reach-1,1
Up Type=0
Dn Type=3
Dn Slope=0.005
Boundary for River Rch & Prof#=LEFT HAND CREEK,Reach-1,2
Up Type=0
Dn Type=3
Dn Slope=0.005
Boundary for River Rch & Prof#=LEFT HAND CREEK,Reach-1,3
Up Type=0
Dn Type=3
Dn Slope=0.005
Boundary for River Rch & Prof#=LEFT HAND CREEK,Reach-1,4
Up Type=0
Dn Type=3
Dn Slope=0.005
Boundary for River Rch & Prof#=LEFT HAND CREEK,Reach-1,5
Up Type=0
Dn Type=3
Dn Slope=0.005
Boundary for River Rch & Prof#=LEFT HAND CREEK,Reach-1,6
Up Type=0
Dn Type=3
Dn Slope=0.005
Boundary for River Rch & Prof#=LEFT HAND CREEK,Reach-1,7
Up Type=0
Dn Type=3
Dn Slope=0.005

--- LEFT HAND CREEK.g01 (geometry) ---

Geom Title=Existing Conditions

River Reach=LEFT HAND CREEK,Reach-1
Reach XY= 30
      2757784.50     10159730.00      2757433.00     10162020.00
      2757839.00     10162861.00      2757532.75     10163827.00
      2757826.50     10164983.00      2757297.75     10166102.00
      2755802.00     10166454.00      2755468.75     10167650.00
      2754710.50     10167421.00      2753879.25     10168490.00
      2753384.75     10168537.00      2752960.50     10168004.00
      2751609.00     10167747.00      2751410.00     10168167.00
      2750668.50     10168063.00      2750109.00     10168692.00
      2749277.50     10168479.00      2748814.50     10169251.00
      2746745.75     10169355.00      2746634.50     10170618.00
      2745956.50     10170805.00      2745382.00     10170553.00
      2744308.50     10171469.00      2744344.00     10172127.00
      2743592.00     10173387.00      2742343.75     10174099.00
      2741004.25     10173894.00      2740305.25     10173186.00
      2739484.75     10173211.00      2738738.25     10173700.00

Type RM Length L Ch R = 1,34000,500,500,500
BEGIN DESCRIPTION:
LEFT HAND CREEK 68.0
END DESCRIPTION:
XS GIS Cut Line= 3
      2757455.67     10159553.08      2757634.20     10160066.11
      2758055.72     10159703.08
#Sta/Elev= 30
  4456.8 1692.71  4622.6 1684.22  4647.4 1683.54  4684.8 1680.95  4746.9 1678.47
  4834.9 1672.04  4866.0 1670.88  4897.1 1668.39  4920.6 1667.47  4954.0 1665.90
  4965.1 1666.23  4993.8 1665.37  4994.0 1664.87  4997.8 1665.37  5038.9 1667.74
  5074.0 1667.73  5088.3 1668.98  5137.7 1670.14  5209.0 1673.75  5251.8 1675.31
  5258.4 1675.00  5272.6 1676.08  5279.2 1675.80  5286.9 1676.77  5322.0 1677.52
  5358.7 1679.35  5421.8 1681.91  5442.7 1681.73  5521.7 1685.80  5556.3 1687.54
#Mann=6,-1,0
  4456.8    0.12       0  4920.6    0.05       0  4993.8    0.05       0
  4997.8    0.05       0  5358.7    0.12       0  5521.7    0.05       0
Bank Sta=4993.8,4997.8
Exp/Cntr=0.3,0.1

Type RM Length L Ch R = 1,33500,500,500,500
BEGIN DESCRIPTION:
LEFT HAND CREEK 67.0
END DESCRIPTION:
XS GIS Cut Line= 3
      2756855.71     10159703.14      2757558.71     10160531.03
      2757805.70     10160353.10
#Sta/Elev= 30
  3913.9 1679.46  3949.6 1677.12  3970.4 1678.75  3984.7 1677.97  4013.3 1674.31
  4034.1 1673.62  4062.7 1670.56  4077.0 1672.47  4091.2 1670.14  4169.2 1677.79
  4183.5 1676.27  4190.1 1677.32  4226.4 1675.48  4247.2 1676.24  4304.3 1671.92
  4425.2 1668.82  4460.3 1665.07  4495.4 1666.87  4524.0 1665.02  4544.8 1665.91
  4630.5 1663.71  4815.1 1664.43  4864.5 1659.57  4893.1 1660.36  4996.1 1651.91
  4996.3 1651.41  5000.1 1651.91  5045.6 1653.99  5181.7 1667.39  5304.4 1671.99
#Mann=3,-1,0
  3913.9    0.05       0  4996.1    0.05       0  5000.1    0.05       0
Bank Sta=4996.1,5000.1
Exp/Cntr=0.3,0.1

Type RM Length L Ch R = 1,33000,500,500,500
BEGIN DESCRIPTION:
LEFT HAND CREEK 66.0
END DESCRIPTION:
XS GIS Cut Line= 3
      2756665.22     10160960.54      2757590.86     10161010.72
      2758005.69     10160653.11
#Sta/Elev= 30
  4073.0 1659.64  4117.2 1657.21  4223.7 1653.21  4323.8 1644.34  4383.9 1640.87
  4398.3 1643.02  4494.1 1646.85  4564.2 1653.03  4644.3 1650.04  4675.1 1653.68
  4757.3 1656.28  4955.8 1649.29  4994.8 1645.33  4999.9 1642.63  5014.1 1639.98
  5014.4 1639.48  5018.1 1639.98  5030.4 1642.79  5051.3 1644.67  5122.6 1645.20
  5164.8 1646.94  5200.5 1649.17  5221.3 1652.94  5257.2 1654.22  5278.4 1657.28
  5321.1 1658.47  5335.4 1660.55  5399.0 1664.35  5491.2 1662.66  5547.7 1666.12
#Mann=6,-1,0
  4073.0    0.12       0  4117.2    0.05       0  4675.1    0.12       0
  4757.3    0.05       0  5014.1    0.05       0  5018.1    0.05       0
Bank Sta=5014.1,5018.1
Exp/Cntr=0.3,0.1

Type RM Length L Ch R = 1,32500,500,500,500
BEGIN DESCRIPTION:
LEFT HAND CREEK 65.0
END DESCRIPTION:
XS GIS Cut Line= 3
      2757123.49     10161432.76      2757600.92     10161454.04
      2757855.71     10161253.09
#Sta/Elev= 30
  4522.1 1635.69  4604.4 1623.40  4614.4 1623.59  4624.4 1621.97  4640.8 1627.25
  4645.8 1625.74  4654.4 1628.00  4694.5 1625.24  4724.5 1628.33  4744.5 1628.88
  4806.6 1627.35  4824.6 1626.51  4854.6 1631.25  4874.6 1632.72  4924.7 1628.44
  4964.7 1628.68  4971.1 1626.91  4984.8 1622.18  4997.9 1621.72  4998.1 1621.22
  5001.9 1621.72  5025.5 1626.17  5031.8 1625.73  5039.9 1627.31  5075.1 1628.92
  5089.6 1631.53  5182.6 1640.65  5224.2 1646.63  5246.7 1648.29  5324.5 1650.28
#Mann=5,-1,0
  4522.1    0.05       0  4806.6    0.12       0  4971.1    0.05       0
  4997.9    0.05       0  5001.9    0.05       0
Bank Sta=4997.9,5001.9
Exp/Cntr=0.3,0.1

Type RM Length L Ch R = 1,32000,500,500,500
BEGIN DESCRIPTION:
LEFT HAND CREEK 64.0
END DESCRIPTION:
XS GIS Cut Line= 3
      2757105.72     10161953.10      2757455.71     10161872.30
      2757705.71     10161803.10
#Sta/Elev= 30
  4640.8 1638.55  4707.5 1626.48  4722.9 1622.35  4757.1 1618.27  4793.0 1613.71
  4798.1 1614.08  4815.2 1611.23  4859.4 1609.34  4917.9 1606.22  4961.8 1605.99
  4979.4 1606.34  4989.7 1600.96  4995.4 1600.30  4995.7 1599.80  4999.4 1600.30
  5055.1 1606.84  5083.0 1612.79  5100.2 1619.85  5101.1 1620.28  5128.9 1625.39
  5145.2 1626.49  5155.6 1628.55  5163.2 1629.09  5168.4 1627.51  5176.4 1629.11
  5197.1 1630.46  5202.7 1633.55  5207.9 1631.66  5228.2 1635.37  5259.4 1635.23
#Mann=8,-1,0
  4640.8    0.12       0  4757.1    0.05       0  4859.4    0.12       0
  4961.8    0.05       0  4995.4    0.05       0  4999.4    0.05       0
  5100.2    0.12       0  5101.1    0.05       0
Bank Sta=4995.4,4999.4
Exp/Cntr=0.3,0.1

Type RM Length L Ch R = 1,31500,500,500,500
BEGIN DESCRIPTION:
LEFT HAND CREEK 63.0
END DESCRIPTION:
XS GIS Cut Line= 3
      2757105.66     10162403.12      2757586.89     10162325.84
      2757705.67     10162103.14
#Sta/Elev= 30
  4512.6 1636.57  4541.1 1630.92  4546.1 1632.27  4573.4 1625.24  4603.0 1620.19
  4675.0 1613.78  4707.8 1609.39  4731.9 1606.41  4816.5 1600.92  4855.7 1599.82
  4958.3 1600.76  4968.4 1598.90  4982.6 1589.71  4982.9 1589.21  4986.6 1589.71
  5004.0 1591.39  5008.4 1593.63  5024.7 1594.06  5030.4 1597.74  5046.7 1599.90
  5059.8 1603.52  5090.6 1600.24  5096.2 1603.38  5112.5 1604.85  5127.8 1604.94
  5140.2 1607.06  5178.4 1607.40  5200.4 1610.06  5216.7 1614.34  5252.4 1618.58
#Mann=4,-1,0
  4512.6    0.12       0  4707.8    0.05       0  4982.6    0.05       0
  4986.6    0.05       0
Bank Sta=4982.6,4986.6
Exp/Cntr=0.3,0.1

Type RM Length L Ch R = 1,31000,500,500,500
BEGIN DESCRIPTION:
LEFT HAND CREEK 62.0
END DESCRIPTION:
XS GIS Cut Line= 3
      2757055.70     10162653.11      2757770.52     10162750.36
      2758005.72     10162703.10
#Sta/Elev= 30
  4278.6 1622.57  4308.9 1622.13  4314.8 1621.62  4319.8 1619.71  4369.4 1617.57
  4410.8 1614.01  4500.6 1608.93  4621.7 1600.48  4687.0 1598.68  4732.7 1594.91
  4752.9 1594.65  4764.4 1593.40  4806.9 1593.13  4884.1 1590.37  4904.2 1585.98
  4934.6 1586.16  4944.7 1587.32  4981.7 1587.26  4986.7 1587.97  5000.0 1587.42
  5005.3 1586.46  5008.9 1584.67  5009.1 1584.17  5012.9 1584.67  5035.9 1592.08
  5046.1 1594.71  5061.8 1597.37  5076.7 1597.35  5178.5 1603.69  5239.9 1608.79
#Mann=6,-1,0
  4278.6    0.12       0  4410.8    0.05       0  4806.9    0.12       0
  5008.9    0.07       0  5012.9    0.12       0  5178.5    0.05       0
Bank Sta=5008.9,5012.9
Exp/Cntr=0.3,0.1

Type RM Length L Ch R = 1,30500,500,500,500
BEGIN DESCRIPTION:
LEFT HAND CREEK 61.0
END DESCRIPTION:
XS GIS Cut Line= 3
      2757067.95     10162842.47      2757818.93     10163224.58
      2758622.11     10163051.13
#Sta/Elev= 30
  4157.4 1607.40  4282.0 1600.46  4334.4 1599.92  4415.5 1595.72  4587.8 1594.20
  4721.3 1588.68  4749.5 1585.96  4804.7 1583.94  4810.3 1582.57  4826.9 1583.06
  4839.3 1585.94  4893.6 1582.02  4982.6 1581.21  5015.1 1576.31  5015.4 1575.81
  5019.1 1576.31  5059.0 1581.05  5075.7 1584.46  5125.0 1587.78  5174.2 1587.93
  5218.4 1590.59  5267.7 1590.81  5360.2 1595.44  5405.2 1597.95  5477.5 1598.92
  5528.7 1602.45  5620.7 1603.03  5682.1 1606.12  5744.9 1611.65  5821.7 1611.41
#Mann=5,-1,0
  4157.4    0.05       0  5015.1    0.05       0  5019.1    0.05       0
  5059.0    0.12       0  5360.2    0.05       0
Bank Sta=5015.1,5019.1
Exp/Cntr=0.3,0.1

Type RM Length L Ch R = 1,30000,500,500,500
BEGIN DESCRIPTION:
LEFT HAND CREEK 60.0
END DESCRIPTION:
XS GIS Cut Line= 3
      2757055.68     10163053.11      2757558.29     10163544.05
      2758505.73     10163303.10
#Sta/Elev= 30
  4297.4 1594.02  4431.8 1587.52  4445.9 1588.33  4537.8 1584.41  4672.3 1583.75
  4778.3 1580.32  4877.3 1579.29  4919.7 1574.62  4926.7 1575.50  4974.3 1571.45
  4974.5 1570.95  4978.3 1571.45  5007.6 1575.54  5059.2 1575.59  5107.3 1578.26
  5174.6 1579.54  5299.1 1582.71  5330.0 1583.71  5469.6 1592.25  5509.5 1596.74
  5533.9 1590.77  5544.2 1590.00  5749.9 1588.90  5790.8 1590.87  5812.5 1589.73
  5843.4 1595.05  5872.7 1596.94  5884.7 1601.40  5930.7 1607.05  5977.6 1610.67
#Mann=9,-1,0
  4297.4    0.05       0  4974.3    0.05       0  4978.3    0.05       0
  5107.3    0.12       0  5174.6    0.05       0  5299.1    0.12       0
  5330.0    0.05       0  5469.6    0.12       0  5930.7    0.05       0
Bank Sta=4974.3,4978.3
Exp/Cntr=0.3,0.1

Type RM Length L Ch R = 1,29500,500,500,500
BEGIN DESCRIPTION:
LEFT HAND CREEK 59.0
END DESCRIPTION:
XS GIS Cut Line= 3
      2757105.72     10163953.12      2757623.88     10164017.98
      2758165.20     10163891.10
#Sta/Elev= 30
  4477.8 1589.38  4503.0 1585.60  4538.2 1581.33  4568.5 1575.45  4602.0 1573.55
  4669.2 1571.29  4762.3 1570.99  4810.3 1573.29  4951.4 1570.33  4971.6 1571.29
  4981.7 1569.27  4989.7 1565.90  4990.0 1565.40  4993.7 1565.90  5022.4 1570.11
  5032.7 1570.32  5073.8 1566.95  5083.0 1570.99  5130.6 1574.41  5248.4 1573.64
  5348.0 1577.97  5390.4 1576.12  5395.5 1573.88  5412.7 1575.44  5438.0 1575.30
  5480.4 1581.59  5485.6 1579.86  5505.1 1581.41  5528.0 1579.78  5556.0 1580.64
#Mann=5,-1,0
  4477.8    0.05       0  4503.0    0.12       0  4602.0    0.05       0
  4989.7    0.05       0  4993.7    0.05       0
Bank Sta=4989.7,4993.7
Exp/Cntr=0.3,0.1

Type RM Length L Ch R = 1,29000,500,500,500
BEGIN DESCRIPTION:
LEFT HAND CREEK 58.0
END DESCRIPTION:
XS GIS Cut Line= 3
      2756866.63     10164474.43      2757795.67     10164448.63
      2758220.74     10164404.99
#Sta/Elev= 30
  4070.6 1583.35  4119.7 1581.16  4269.7 1576.64  4359.8 1573.02  4409.8 1572.35
  4439.8 1570.73  4489.8 1570.19  4529.8 1567.70  4539.8 1568.97  4599.9 1566.91
  4661.6 1566.03  4769.9 1566.53  4880.0 1566.07  4920.0 1566.81  4960.0 1565.84
  4990.0 1564.36  5002.5 1563.56  5003.0 1562.49  5003.3 1561.99  5006.8 1561.99
  5007.0 1562.49  5060.3 1568.69  5110.6 1571.10  5150.8 1572.25  5241.3 1573.10
  5297.7 1575.96  5302.7 1575.69  5391.9 1578.95  5422.2 1580.44  5427.3 1581.22
#Mann=3,-1,0
  4070.6    0.05       0  5003.0    0.05       0  5007.0    0.05       0
Bank Sta=5003,5007
Exp/Cntr=0.3,0.1

Type RM Length L Ch R = 1,28500,500,500,500
BEGIN DESCRIPTION:
LEFT HAND CREEK 57.0
END DESCRIPTION:
XS GIS Cut Line= 3
      2756901.30     10164766.10      2757735.59     10164877.51
      2758255.72     10164753.10
#Sta/Elev= 30
  4158.3 1575.76  4243.4 1573.87  4414.9 1567.01  4624.3 1561.88  4636.9 1560.36
  4667.2 1561.53  4707.5 1561.10  4737.8 1561.90  4959.7 1563.68  4969.8 1563.61
  4979.9 1562.46  4995.5 1558.90  4995.8 1558.40  4999.5 1558.90  5010.4 1559.70
  5020.7 1562.17  5043.4 1562.93  5061.8 1562.26  5092.6 1563.78  5144.0 1563.69
  5205.7 1564.77  5300.9 1569.63  5385.0 1574.59  5427.0 1578.31  5432.2 1577.86
  5469.1 1580.71  5483.4 1580.82  5511.2 1583.04  5516.3 1582.73  5534.8 1584.00
#Mann=3,-1,0
  4158.3    0.05       0  4995.5    0.05       0  4999.5    0.05       0
Bank Sta=4995.5,4999.5
Exp/Cntr=0.3,0.1

Type RM Length L Ch R = 1,28000,418,418,418
BEGIN DESCRIPTION:
LEFT HAND CREEK 56.0
END DESCRIPTION:
XS GIS Cut Line= 3
      2756942.96     10165064.70      2757689.59     10165290.76
      2758441.81     10165314.67
#Sta/Elev= 30
  4219.9 1563.78  4437.8 1558.10  4503.7 1555.60  4513.3 1554.14  4513.6 1553.64
  4517.3 1554.14  4588.4 1556.99  4766.1 1558.64  4881.0 1557.98  4901.9 1557.34
  4919.7 1555.06  4933.2 1555.19  4964.6 1559.79  4985.5 1555.11  4990.8 1555.03
  5016.1 1555.71  5036.1 1558.98  5056.1 1560.83  5206.2 1564.02  5236.3 1561.86
  5276.2 1561.93  5326.3 1558.40  5356.3 1561.43  5386.3 1560.36  5406.3 1561.75
  5466.3 1562.30  5536.4 1567.38  5695.4 1572.35  5742.7 1574.22  5752.6 1574.85
#Mann=5,-1,0
  4219.9    0.05       0  4513.3    0.05       0  4517.3    0.05       0
  5695.4    0.12       0  5742.7    0.05       0
Bank Sta=4513.3,4517.3
Exp/Cntr=0.3,0.1

Type RM Length L Ch R = 1,27582,582,582,582
BEGIN DESCRIPTION:
LEFT HAND CREEK 55.0
END DESCRIPTION:
XS GIS Cut Line= 3
      2757016.13     10165232.87      2757443.91     10165594.57
      2758483.18     10165657.83
#Sta/Elev= 30
  4439.8 1558.87  4599.8 1554.80  4623.3 1554.62  4645.3 1551.13  4680.5 1553.66
  4760.2 1553.40  4841.4 1553.88  4966.1 1551.97  4992.5 1551.39  5014.5 1547.58
  5035.4 1548.56  5061.9 1547.13  5062.2 1546.63  5065.9 1547.13  5070.5 1549.10
  5075.5 1547.36  5099.4 1547.19  5135.2 1550.92  5230.5 1550.85  5257.3 1551.70
  5319.8 1552.75  5359.9 1550.63  5400.0 1555.70  5450.1 1552.38  5490.1 1554.98
  5590.3 1556.49  5670.5 1560.95  5979.7 1570.64  6028.0 1572.59  6041.2 1573.01
#Mann=11,-1,0
  4439.8    0.05       0  4599.8    0.12       0  4760.2    0.05       0
  4841.4    0.12       0  4966.1    0.05       0  5061.9    0.05       0
  5065.9    0.05       0  5230.5    0.12       0  5257.3    0.05       0
  5979.7    0.12       0  6028.0    0.05       0
Bank Sta=5061.9,5065.9
Exp/Cntr=0.3,0.1

Type RM Length L Ch R = 1,27000,500,500,500
BEGIN DESCRIPTION:
LEFT HAND CREEK 54.0
END DESCRIPTION:
XS GIS Cut Line= 3
      2756655.67     10165053.09      2757359.38     10166032.73
      2757605.67     10166453.09
#Sta/Elev= 30
  3793.8 1568.31  4038.1 1558.39  4079.9 1555.26  4088.5 1555.24  4094.6 1556.55
  4124.1 1556.12  4323.3 1550.04  4346.3 1548.41  4381.9 1550.50  4446.4 1551.14
  4503.5 1550.54  4524.4 1551.27  4553.8 1550.29  4618.8 1551.04  4790.8 1547.22
  4796.9 1547.90  4926.6 1546.65  4954.1 1547.30  4983.5 1546.28  4995.2 1543.24
  4995.4 1542.74  4999.2 1543.24  5006.9 1543.86  5025.9 1545.57  5037.2 1545.50
  5047.4 1546.87  5143.2 1553.02  5201.8 1555.92  5406.1 1562.44  5487.2 1563.39
#Mann=5,-1,0
  3793.8    0.05       0  4995.2    0.05       0  4999.2    0.05       0
  5006.9    0.12       0  5037.2    0.05       0
Bank Sta=4995.2,4999.2
Exp/Cntr=0.3,0.1

Type RM Length L Ch R = 1,26500,500,500,500
BEGIN DESCRIPTION:
LEFT HAND CREEK 53.0
END DESCRIPTION:
XS GIS Cut Line= 3
      2756555.67     10165253.09      2756968.42     10166261.70
      2757355.65     10166503.09
#Sta/Elev= 30
  3910.2 1561.66  3996.7 1559.71  4192.0 1552.19  4394.9 1546.11  4424.3 1543.67
  4472.1 1543.25  4547.7 1545.48  4590.9 1545.55  4632.5 1544.79  4637.9 1545.34
  4661.9 1544.39  4667.3 1545.21  4709.8 1543.96  4753.0 1544.30  4870.2 1542.06
  4947.5 1542.56  4977.0 1541.17  4988.7 1537.70  4989.0 1537.20  4992.7 1537.70
  5007.4 1538.50  5013.3 1540.40  5020.3 1541.15  5049.9 1543.04  5173.5 1547.76
  5196.2 1549.66  5406.2 1556.22  5427.4 1560.19  5433.3 1559.28  5456.3 1560.58
#Mann=3,-1,0
  3910.2    0.05       0  4988.7    0.05       0  4992.7    0.05       0
Bank Sta=4988.7,4992.7
Exp/Cntr=0.3,0.1

Type RM Length L Ch R = 1,26000,500,500,500
BEGIN DESCRIPTION:
LEFT HAND CREEK 52.0
END DESCRIPTION:
XS GIS Cut Line= 3
      2756255.68     10165353.10      2756517.04     10166372.63
      2756405.69     10167003.07
#Sta/Elev= 30
  3947.5 1562.51  3999.1 1561.14  4128.5 1553.81  4195.3 1552.48  4215.9 1549.93
  4257.2 1551.28  4368.0 1547.45  4373.1 1548.30  4432.7 1548.41  4525.6 1546.63
  4531.1 1545.68  4571.9 1544.93  4701.1 1537.64  4735.0 1538.03  4742.4 1537.12
  4763.1 1538.34  4794.0 1538.56  4852.2 1536.75  4933.8 1538.43  4974.5 1537.31
  4995.7 1533.29  4995.9 1532.79  4999.7 1533.29  5010.6 1535.40  5031.0 1535.73
  5041.4 1537.43  5071.6 1539.26  5327.3 1544.98  5569.2 1554.76  5640.2 1558.80
#Mann=3,-1,0
  3947.5    0.05       0  4995.7    0.05       0  4999.7    0.05       0
Bank Sta=4995.7,4999.7
Exp/Cntr=0.3,0.1

Type RM Length L Ch R = 1,25500,500,500,500
BEGIN DESCRIPTION:
LEFT HAND CREEK 51.0
END DESCRIPTION:
XS GIS Cut Line= 3
      2756005.69     10165953.15      2756039.96     10166320.36
      2756405.69     10167103.13
#Sta/Elev= 30
  4631.2 1553.83  4680.7 1549.80  4685.7 1550.31  4691.4 1549.28  4751.7 1545.40
  4892.3 1538.38  4922.4 1538.00  4962.6 1535.15  4990.6 1531.70  4990.9 1531.20
  4994.8 1531.70  5014.1 1533.51  5036.2 1533.96  5073.7 1533.60  5113.4 1534.77
  5214.3 1534.08  5262.0 1535.13  5376.2 1539.52  5389.4 1540.69  5488.7 1543.72
  5610.1 1549.52  5752.9 1556.96  5786.8 1562.17  5797.8 1562.84  5804.1 1563.11
  5809.6 1561.93  5819.8 1563.84  5841.9 1563.18  5849.8 1562.12  5864.0 1562.55
#Mann=3,-1,0
  4631.2    0.05       0  4990.6    0.05       0  4994.8    0.05       0
Bank Sta=4990.6,4994.8
Exp/Cntr=0.3,0.1

Type RM Length L Ch R = 1,25000,500,500,500
BEGIN DESCRIPTION:
LEFT HAND CREEK 50.0
END DESCRIPTION:
XS GIS Cut Line= 3
      2755463.82     10165995.29      2755783.49     10166660.80
      2756205.66     10167053.09
#Sta/Elev= 30
  4261.7 1540.47  4389.9 1538.07  4536.9 1536.65  4735.1 1532.72  4780.4 1532.94
  4791.8 1532.03  4831.2 1531.46  4936.0 1531.79  4950.0 1530.77  4967.1 1530.95
  4972.6 1528.91  4989.7 1529.37  4996.4 1527.32  4996.7 1526.82  5000.6 1527.32
  5017.1 1527.65  5024.5 1529.93  5058.8 1530.34  5109.5 1531.61  5218.7 1536.29
  5229.7 1537.80  5236.5 1537.31  5279.0 1538.88  5314.7 1541.11  5321.5 1540.71
  5420.7 1545.95  5434.9 1546.09  5463.2 1548.65  5498.4 1548.30  5576.3 1550.64
#Mann=5,-1,0
  4261.7    0.05       0  4996.4    0.05       0  5000.6    0.05       0
  5058.8    0.12       0  5218.7    0.05       0
Bank Sta=4996.4,5000.6
Exp/Cntr=0.3,0.1

Type RM Length L Ch R = 1,24500,500,500,500
BEGIN DESCRIPTION:
LEFT HAND CREEK 49.0
END DESCRIPTION:
XS GIS Cut Line= 3
      2755155.68     10166203.09      2755565.32     10167070.09
      2756355.73     10167103.11
#Sta/Elev= 30
  4041.1 1545.10  4207.0 1537.97  4339.7 1534.02  4379.5 1533.99  4402.3 1535.60
  4453.3 1536.30  4470.6 1535.67  4498.8 1536.64  4516.1 1535.64  4521.6 1536.78
  4544.4 1534.64  4612.7 1533.09  4732.0 1532.25  4749.0 1533.16  4800.3 1531.61
  4874.1 1527.79  4903.8 1527.82  4936.9 1524.85  4996.7 1522.97  4997.0 1522.47
  5001.1 1522.97  5030.4 1525.69  5080.4 1527.64  5180.5 1528.20  5320.6 1533.43
  5433.7 1539.42  5470.8 1542.49  5673.6 1551.75  5731.0 1556.34  5791.1 1559.44
#Mann=3,-1,0
  4041.1    0.05       0  4996.7    0.05       0  5001.1    0.05       0
Bank Sta=4996.7,5001.1
Exp/Cntr=0.3,0.1

Type RM Length L Ch R = 1,24000,500,500,500
BEGIN DESCRIPTION:
LEFT HAND CREEK 48.0
END DESCRIPTION:
XS GIS Cut Line= 3
      2755205.70     10167103.13      2755404.02     10167435.81
      2756205.66     10167353.11
#Sta/Elev= 30
  4612.7 1530.47  4620.5 1528.98  4626.3 1529.50  4641.9 1527.24  4663.3 1527.05
  4678.9 1525.48  4684.7 1525.96  4737.3 1523.74  4743.1 1524.34  4774.3 1523.22
  4812.5 1523.53  4896.9 1524.62  4976.7 1524.18  4992.3 1523.22  4996.7 1520.97
  5011.7 1520.15  5031.8 1521.70  5041.9 1523.51  5071.0 1524.13  5073.8 1519.64
  5074.1 1519.14  5078.2 1519.64  5095.3 1520.14  5102.2 1520.25  5122.3 1523.51
  5152.5 1525.56  5283.2 1526.25  5467.0 1530.32  5604.9 1535.26  5805.9 1543.83
#Mann=5,-1,0
  4612.7    0.05       0  4812.5    0.12       0  5073.8    0.07       0
  5078.2    0.12       0  5095.3    0.05       0
Bank Sta=5073.8,5078.2
Exp/Cntr=0.3,0.1

Type RM Length L Ch R = 1,23500,500,500,500
BEGIN DESCRIPTION:
LEFT HAND CREEK 47.0
END DESCRIPTION:
XS GIS Cut Line= 3
      2755055.69     10166203.14      2755243.01     10167609.92
      2755305.69     10168103.15
#Sta/Elev= 30
  3580.8 1544.45  3974.2 1533.40  4105.4 1533.14  4125.5 1531.53  4155.8 1531.85
  4223.1 1529.39  4246.6 1530.90  4287.0 1530.08  4307.1 1532.12  4337.4 1531.58
  4357.6 1532.77  4367.7 1531.72  4387.8 1533.04  4418.1 1529.90  4458.5 1529.92
  4478.6 1527.63  4488.7 1528.18  4525.9 1525.30  4660.2 1521.78  4755.6 1521.38
  4907.0 1522.32  4942.7 1521.14  4955.1 1519.15  4990.5 1515.42  4990.9 1514.92
  4995.8 1515.42  4999.1 1516.38  5033.5 1516.58  5059.8 1520.66  5497.2 1536.09
#Mann=5,-1,0
  3580.8    0.05       0  4755.6    0.12       0  4955.1    0.05       0
  4990.5    0.03       0  4995.8    0.05       0
Bank Sta=4990.5,4995.8
Exp/Cntr=0.3,0.1

Type RM Length L Ch R = 1,23000,500,500,500
BEGIN DESCRIPTION:
LEFT HAND CREEK 46.0
END DESCRIPTION:
XS GIS Cut Line= 3
      2754105.66     10166603.08      2754811.01     10167433.82
      2755305.66     10168253.07
#Sta/Elev= 30
  3910.2 1541.74  4329.3 1528.85  4506.1 1526.12  4563.2 1526.14  4776.1 1521.21
  4875.2 1517.44  4910.3 1517.19  4924.6 1516.34  4932.3 1514.36  4938.9 1514.02
  4946.6 1513.66  4953.1 1515.01  4957.0 1513.38  4957.4 1512.88  4962.4 1513.38
  4988.3 1514.00  4996.0 1515.11  5002.5 1513.62  5017.7 1516.22  5039.1 1515.53
  5069.3 1517.87  5198.2 1519.90  5330.2 1520.36  5578.6 1527.06  5774.6 1534.43
  5898.6 1540.66  5933.8 1542.93  5943.4 1544.49  5949.3 1543.82  5957.0 1544.52
#Mann=3,-1,0
  3910.2    0.05       0  4957.0    0.05       0  4962.4    0.05       0
Bank Sta=4957,4962.4
Exp/Cntr=0.3,0.1

Type RM Length L Ch R = 1,22500,500,500,500
BEGIN DESCRIPTION:
LEFT HAND CREEK 45.0
END DESCRIPTION:
XS GIS Cut Line= 3
      2754105.67     10166853.09      2754499.33     10167697.98
      2755305.65     10168353.09
#Sta/Elev= 30
  4067.9 1537.74  4277.5 1528.23  4339.2 1526.51  4407.8 1526.82  4436.2 1528.77
  4453.6 1527.78  4459.1 1528.24  4504.8 1526.90  4608.5 1525.64  4647.6 1524.13
  4818.7 1522.32  4972.6 1514.54  4978.8 1511.75  4984.3 1510.69  5005.5 1509.79
  5005.9 1509.29  5010.9 1509.79  5021.8 1511.55  5029.7 1511.96  5036.2 1513.34
  5085.7 1516.47  5349.4 1518.06  5477.2 1521.31  5512.4 1522.67  5520.3 1523.55
  5619.4 1526.62  5903.9 1541.71  5974.5 1546.09  6002.2 1546.92  6038.9 1547.75
#Mann=4,-1,0
  4067.9    0.05       0  5005.5    0.05       0  5010.9    0.05       0
  6002.2    0.12       0
Bank Sta=5005.5,5010.9
Exp/Cntr=0.3,0.1

Type RM Length L Ch R = 1,22000,500,500,500
BEGIN DESCRIPTION:
LEFT HAND CREEK 44.0
END DESCRIPTION:
XS GIS Cut Line= 3
      2754005.68     10167003.09      2754116.00     10167982.60
      2755055.67     10168503.10
#Sta/Elev= 30
  4014.3 1530.16  4024.4 1529.20  4125.0 1525.44  4265.9 1522.53  4316.2 1522.62
  4329.2 1521.99  4346.4 1522.59  4396.7 1522.42  4509.1 1524.99  4608.1 1524.89
  4789.2 1517.18  4819.4 1515.05  4858.9 1516.57  4863.9 1515.02  4879.8 1515.73
  4899.9 1513.14  4953.9 1511.83  4995.0 1506.85  4995.4 1506.35  5000.5 1506.85
  5008.4 1507.40  5014.1 1509.25  5022.5 1510.34  5057.6 1512.54  5205.4 1514.34
  5323.2 1514.54  5448.0 1516.86  5479.8 1516.81  5913.9 1531.31  6074.2 1537.57
#Mann=3,-1,0
  4014.3    0.05       0  4995.0    0.05       0  5000.5    0.05       0
Bank Sta=4995,5000.5
Exp/Cntr=0.3,0.1

Type RM Length L Ch R = 1,21500,500,500,500
BEGIN DESCRIPTION:
LEFT HAND CREEK 43.0
END DESCRIPTION:
XS GIS Cut Line= 3
      2753831.86     10167891.09      2753963.14     10168349.56
      2754137.41     10168925.79
#Sta/Elev= 30
  4523.1 1520.14  4681.2 1520.93  4771.4 1518.97  4776.6 1517.93  4849.3 1514.84
  4883.1 1514.50  4889.3 1515.45  4910.1 1515.67  4922.0 1513.95  4950.6 1512.18
  4972.5 1509.49  4994.8 1505.46  5020.0 1505.33  5020.4 1504.83  5025.5 1505.33
  5027.9 1507.44  5035.0 1507.84  5087.3 1507.72  5099.0 1508.50  5132.0 1507.70
  5139.5 1505.69  5170.9 1509.82  5191.8 1510.95  5203.1 1512.75  5307.2 1517.01
  5367.8 1517.38  5373.0 1518.19  5438.9 1519.03  5452.9 1520.16  5602.0 1522.60
#Mann=3,-1,0
  4523.1    0.05       0  5020.0    0.05       0  5025.5    0.05       0
Bank Sta=5020,5025.5
Exp/Cntr=0.3,0.1

Type RM Length L Ch R = 1,21000,500,500,500
BEGIN DESCRIPTION:
LEFT HAND CREEK 42.0
END DESCRIPTION:
XS GIS Cut Line= 3
      2753776.30     10167821.67      2753575.26     10168469.18
      2753200.31     10169133.47
#Sta/Elev= 30
  4322.0 1518.82  4372.7 1519.65  4410.5 1518.24  4522.5 1521.73  4573.3 1520.96
  4811.7 1512.35  4817.0 1510.68  4849.6 1508.68  4952.5 1505.09  4976.7 1501.63
  4977.2 1501.13  4983.0 1501.63  5047.4 1505.66  5061.9 1504.33  5090.7 1505.62
  5112.3 1510.77  5149.9 1511.04  5171.5 1509.18  5177.3 1507.48  5214.9 1507.19
  5274.1 1508.82  5370.9 1514.31  5419.9 1514.32  5509.8 1517.33  5613.1 1521.97
  5635.2 1525.58  5662.6 1524.71  5716.0 1532.95  5727.9 1531.87  5762.8 1532.59
#Mann=3,-1,0
  4322.0    0.05       0  4976.7    0.05       0  4983.0    0.05       0
Bank Sta=4976.7,4983
Exp/Cntr=0.3,0.1

Type RM Length L Ch R = 1,20500,500,500,500
BEGIN DESCRIPTION:
LEFT HAND CREEK 41.0
END DESCRIPTION:
XS GIS Cut Line= 3
      2753699.95     10167703.56      2753199.25     10168351.69
      2752734.62     10169043.91
#Sta/Elev= 30
  4181.0 1516.56  4411.5 1515.36  4461.3 1513.70  4483.7 1514.90  4589.9 1512.86
  4660.6 1509.08  4683.2 1509.85  4704.0 1507.07  4724.8 1508.93  4747.5 1509.04
  4789.2 1504.18  4897.0 1505.08  4993.4 1499.45  4993.9 1498.95  4999.8 1499.45
  5032.6 1500.70  5038.6 1503.87  5074.6 1506.15  5419.4 1514.55  5449.7 1513.74
  5472.1 1515.50  5530.7 1517.54  5652.1 1516.72  5659.7 1518.06  5724.3 1519.67
  5752.7 1524.96  5782.7 1525.23  5788.8 1523.77  5809.8 1522.75  5833.7 1524.99
#Mann=5,-1,0
  4181.0    0.05       0  4993.4    0.05       0  4999.8    0.05       0
  5419.4    0.12       0  5472.1    0.05       0
Bank Sta=4993.4,4999.8
Exp/Cntr=0.3,0.1

Type RM Length L Ch R = 1,20000,500,500,500
BEGIN DESCRIPTION:
LEFT HAND CREEK 40.0
END DESCRIPTION:
XS GIS Cut Line= 3
      2753470.75     10167349.43      2752906.48     10167982.85
      2752346.24     10168938.89
#Sta/Elev= 30
  4151.7 1514.34  4236.1 1512.44  4278.0 1513.04  4299.7 1510.10  4356.5 1507.54
  4391.7 1508.70  4405.9 1510.56  4412.6 1513.01  4420.1 1513.00  4434.3 1511.93
  4441.0 1508.98  4469.4 1508.14  4526.3 1510.27  4547.2 1508.39  4646.7 1506.03
  4732.0 1505.11  4767.1 1506.22  4838.7 1503.76  4841.9 1503.84  4951.0 1500.35
  4987.0 1496.36  5005.5 1496.10  5006.0 1495.60  5012.0 1496.10  5067.4 1498.54
  5126.1 1497.08  5336.4 1499.37  5498.7 1502.97  5834.8 1512.72  6108.1 1524.30
#Mann=5,-1,0
  4151.7    0.05       0  4838.7    0.12       0  4841.9    0.05       0
  5005.5    0.05       0  5012.0    0.05       0
Bank Sta=5005.5,5012
Exp/Cntr=0.3,0.1

Type RM Length L Ch R = 1,19500,500,500,500
BEGIN DESCRIPTION:
LEFT HAND CREEK 39.0
END DESCRIPTION:
XS GIS Cut Line= 3
      2753255.69     10167253.11      2752453.13     10167815.34
      2752055.69     10168753.09
#Sta/Elev= 30
  4020.1 1515.11  4056.7 1514.56  4063.3 1512.48  4084.2 1510.89  4105.6 1512.07
  4119.9 1511.17  4142.2 1513.08  4214.9 1511.96  4364.0 1507.26  4414.6 1508.56
  4465.1 1507.54  4602.0 1507.46  4679.6 1505.32  4759.8 1500.56  4896.7 1496.81
  4923.7 1494.55  4947.2 1494.13  4960.3 1495.28  5001.3 1492.59  5001.8 1492.09
  5007.9 1492.59  5028.3 1494.21  5041.0 1493.99  5057.4 1496.15  5110.2 1494.67
  5286.8 1501.99  5529.8 1510.02  5768.7 1514.58  5942.5 1520.18  6018.5 1524.10
#Mann=3,-1,0
  4020.1    0.05       0  5001.3    0.05       0  5007.9    0.05       0
Bank Sta=5001.3,5007.9
Exp/Cntr=0.3,0.1

Type RM Length L Ch R = 1,19000,500,500,500
BEGIN DESCRIPTION:
LEFT HAND CREEK 38.0
END DESCRIPTION:
XS GIS Cut Line= 3
      2752055.68     10167103.12      2752003.85     10167809.42
      2751955.69     10168203.08
#Sta/Elev= 30
  4291.8 1507.27  4321.9 1507.73  4402.1 1505.78  4492.0 1500.78  4602.6 1497.04
  4672.8 1496.34  4722.9 1494.60  4753.0 1495.63  4846.6 1492.49  4883.4 1492.53
  4953.6 1490.15  4994.8 1485.85  4995.3 1485.35  5003.8 1485.85  5013.8 1486.30
  5022.5 1488.52  5027.5 1487.34  5038.9 1489.69  5054.1 1491.86  5074.2 1493.35
  5134.7 1496.37  5185.1 1499.95  5190.4 1503.82  5195.5 1501.78  5215.3 1504.43
  5235.4 1503.70  5265.7 1504.29  5295.9 1502.61  5316.0 1502.74  5396.6 1507.11
#Mann=5,-1,0
  4291.8    0.05       0  4846.6    0.12       0  4994.8    0.07       0
  5003.8    0.12       0  5038.9    0.05       0
Bank Sta=4994.8,5003.8
Exp/Cntr=0.3,0.1

Type RM Length L Ch R = 1,18500,500,500,500
BEGIN DESCRIPTION:
LEFT HAND CREEK 37.0
END DESCRIPTION:
XS GIS Cut Line= 3
      2751605.69     10166803.10      2751545.39     10167806.89
      2751805.70     10168203.13
#Sta/Elev= 30
  3994.4 1506.40  4134.7 1501.75  4295.0 1499.08  4395.1 1495.74  4545.4 1493.78
  4665.6 1494.11  4845.9 1491.55  4896.0 1488.11  4911.4 1484.97  4926.1 1485.21
  4936.1 1487.28  4976.2 1483.42  5005.6 1483.20  5032.6 1485.02  5047.7 1484.72
  5058.1 1482.91  5058.6 1482.41  5067.4 1482.91  5077.9 1483.23  5091.2 1487.09
  5104.9 1488.78  5279.7 1492.45  5315.9 1495.61  5337.0 1494.38  5366.4 1496.72
  5379.1 1496.31  5394.2 1499.08  5409.3 1499.17  5445.5 1503.84  5474.1 1505.18
#Mann=3,-1,0
  3994.4    0.05       0  5058.1    0.05       0  5067.4    0.05       0
Bank Sta=5058.1,5067.4
Exp/Cntr=0.3,0.1

Type RM Length L Ch R = 1,18000,500,500,500
BEGIN DESCRIPTION:
LEFT HAND CREEK 36.0
END DESCRIPTION:
XS GIS Cut Line= 3
      2751105.69     10167103.16      2751317.10     10168214.33
      2751705.69     10168453.12
#Sta/Elev= 30
  3868.9 1503.04  4062.3 1498.12  4322.7 1493.23  4541.7 1491.48  4693.2 1488.03
  4927.5 1487.67  4947.9 1487.00  4964.4 1483.97  4969.5 1484.15  4978.4 1481.90
  4988.6 1481.74  4992.1 1480.64  4992.6 1480.14  5001.5 1480.64  5021.1 1482.08
  5033.6 1481.79  5042.4 1482.58  5048.3 1484.29  5085.0 1486.86  5137.1 1487.64
  5143.0 1488.55  5186.1 1488.70  5274.4 1495.96  5332.4 1498.02  5369.1 1502.35
  5390.4 1503.35  5427.1 1508.80  5433.0 1508.70  5453.2 1514.25  5456.1 1514.25
#Mann=3,-1,0
  3868.9    0.05       0  4992.1    0.05       0  5001.5    0.05       0
Bank Sta=4992.1,5001.5
Exp/Cntr=0.3,0.1

Type RM Length L Ch R = 1,17500,500,500,500
BEGIN DESCRIPTION:
LEFT HAND CREEK 35.0
END DESCRIPTION:
XS GIS Cut Line= 3
      2751055.68     10167103.14      2750842.78     10168100.26
      2751105.71     10168503.15
#Sta/Elev= 30
  3980.4 1504.19  4368.9 1491.77  4542.8 1490.10  4563.2 1489.12  4573.4 1487.54
  4583.9 1489.28  4593.9 1489.29  4634.8 1487.42  4685.9 1488.50  4771.7 1487.33
  4849.5 1483.93  4880.2 1478.62  4890.4 1478.16  4900.7 1478.07  4910.0 1479.35
  4931.3 1478.87  4951.8 1479.78  4972.2 1477.95  4982.5 1478.49  5013.2 1477.62
  5013.7 1477.12  5022.6 1477.62  5048.1 1480.08  5206.4 1485.52  5235.1 1485.76
  5322.7 1490.75  5364.9 1492.21  5380.0 1493.84  5416.2 1495.74  5481.1 1498.03
#Mann=3,-1,0
  3980.4    0.05       0  5013.2    0.05       0  5022.6    0.05       0
Bank Sta=5013.2,5022.6
Exp/Cntr=0.3,0.1

Type RM Length L Ch R = 1,17000,500,500,500
BEGIN DESCRIPTION:
LEFT HAND CREEK 34.0
END DESCRIPTION:
XS GIS Cut Line= 3
      2750330.69     10168028.12      2750461.94     10168290.41
      2751255.70     10168653.12
#Sta/Elev= 30
  4706.7 1484.89  4723.6 1484.59  4768.2 1484.58  4868.8 1481.61  4885.5 1481.90
  4924.7 1480.10  4946.3 1477.98  4958.3 1477.01  4969.4 1477.30  4995.3 1472.71
  4995.8 1472.21  5004.8 1472.71  5059.1 1474.20  5071.1 1478.30  5088.6 1480.50
  5147.0 1482.58  5283.8 1482.55  5479.0 1488.75  5496.6 1490.29  5502.1 1490.01
  5564.8 1493.49  5594.2 1496.26  5599.7 1495.83  5668.7 1499.72  5812.4 1510.83
  5817.9 1510.14  5828.7 1510.86  5835.4 1512.20  5840.9 1511.32  5872.7 1512.60
#Mann=5,-1,0
  4706.7    0.05       0  4723.6    0.12       0  4946.3    0.05       0
  4995.3    0.03       0  5004.8    0.05       0
Bank Sta=4995.3,5004.8
Exp/Cntr=0.3,0.1

Type RM Length L Ch R = 1,16500,500,500,500
BEGIN DESCRIPTION:
LEFT HAND CREEK 33.0
END DESCRIPTION:
XS GIS Cut Line= 3
      2749755.70     10167953.14      2750153.39     10168674.59
      2751105.67     10169453.10
#Sta/Elev= 30
  4176.2 1496.09  4189.9 1496.29  4227.8 1493.73  4461.6 1484.69  4662.2 1479.59
  4874.3 1478.05  4933.9 1475.79  4955.7 1474.12  4964.1 1472.48  4986.9 1471.44
  4987.6 1470.41  4988.1 1469.91  4999.4 1470.41  5015.4 1473.07  5028.8 1477.23
  5057.0 1479.38  5341.3 1480.08  5370.0 1481.43  5384.4 1480.91  5491.3 1483.19
  5512.2 1484.45  5576.0 1484.99  5661.7 1487.76  5938.6 1493.03  5952.9 1494.41
  6080.7 1499.68  6115.9 1502.36  6130.2 1504.65  6159.0 1503.24  6230.0 1508.43
#Mann=3,-1,0
  4176.2    0.05       0  4987.6    0.03       0  4999.4    0.05       0
Bank Sta=4987.6,4999.4
Exp/Cntr=0.3,0.1

Type RM Length L Ch R = 1,16000,500,500,500
BEGIN DESCRIPTION:
LEFT HAND CREEK 32.0
END DESCRIPTION:
XS GIS Cut Line= 3
      2749655.68     10168203.10      2749690.37     10168535.60
      2750067.98     10169432.77
#Sta/Elev= 30
  4665.7 1488.66  4805.9 1481.69  4810.9 1482.04  4876.8 1478.26  4937.2 1476.73
  4967.3 1475.26  4977.4 1473.50  4987.4 1470.57  4996.2 1469.03  5013.1 1468.39
  5013.6 1467.89  5024.4 1467.89  5024.9 1468.39  5025.5 1469.76  5030.9 1468.90
  5040.7 1472.87  5062.4 1473.92  5078.4 1473.51  5107.6 1475.40  5149.2 1476.49
  5170.9 1476.31  5192.6 1477.19  5361.2 1476.93  5461.6 1475.07  5514.5 1474.95
  5637.4 1476.69  5797.3 1477.85  5832.7 1479.01  5926.9 1479.28  5973.4 1480.22
#Mann=3,-1,0
  4665.7    0.05       0  5013.1    0.05       0  5024.9    0.05       0
Bank Sta=5013.1,5024.9
Exp/Cntr=0.3,0.1

Type RM Length L Ch R = 1,15500,500,500,500
BEGIN DESCRIPTION:
LEFT HAND CREEK 31.0
END DESCRIPTION:
XS GIS Cut Line= 3
      2748762.40     10168085.52      2749215.93     10168520.34
      2749984.66     10169432.78
#Sta/Elev= 30
  4371.7 1483.37  4435.9 1482.62  4492.5 1478.16  4528.1 1477.45  4549.1 1479.30
  4570.2 1476.41  4626.8 1474.97  4634.0 1476.11  4641.0 1474.65  4648.2 1476.81
  4655.1 1475.07  4662.3 1476.84  4669.3 1475.52  4676.5 1477.53  4704.8 1477.80
  4740.0 1476.08  4818.0 1477.08  4916.8 1475.58  4980.6 1470.03  4992.5 1466.82
  4993.0 1466.32  5004.3 1466.82  5072.5 1472.80  5150.5 1474.46  5363.8 1473.50
  5583.6 1477.18  5626.5 1472.23  5655.1 1472.08  5696.7 1474.74  6193.1 1478.43
#Mann=3,-1,0
  4371.7    0.05       0  4992.5    0.05       0  5004.3    0.05       0
Bank Sta=4992.5,5004.3
Exp/Cntr=0.3,0.1

Type RM Length L Ch R = 1,15000,500,500,500
BEGIN DESCRIPTION:
LEFT HAND CREEK 30.0
END DESCRIPTION:
XS GIS Cut Line= 3
      2748205.69     10168553.12      2749044.84     10168967.08
      2750005.68     10169903.11
#Sta/Elev= 30
  4064.3 1485.95  4347.7 1479.61  4566.1 1471.66  4622.7 1471.13  4684.5 1472.49
  4789.1 1470.22  4931.5 1471.29  4959.5 1470.04  4976.4 1465.89  4991.4 1464.84
  4991.9 1464.34  5003.9 1464.84  5019.0 1465.57  5026.1 1467.28  5068.6 1469.43
  5111.0 1468.40  5181.7 1470.98  5287.7 1468.79  5379.6 1473.77  5407.9 1474.75
  5415.0 1473.84  5436.2 1475.87  5443.3 1474.88  5450.3 1476.71  5478.6 1476.10
  5549.3 1478.53  5634.2 1479.16  5832.3 1477.71  6150.4 1483.94  6341.4 1485.73
#Mann=3,-1,0
  4064.3    0.05       0  4991.4    0.05       0  5003.9    0.05       0
Bank Sta=4991.4,5003.9
Exp/Cntr=0.3,0.1

Type RM Length L Ch R = 1,14500,500,500,500
BEGIN DESCRIPTION:
LEFT HAND CREEK 29.0
END DESCRIPTION:
XS GIS Cut Line= 3
      2748155.69     10168553.11      2748708.05     10169277.05
      2749055.70     10170203.15
#Sta/Elev= 30
  4089.4 1486.43  4217.3 1484.46  4389.7 1478.13  4460.4 1476.91  4524.8 1474.52
  4581.0 1475.02  4639.1 1472.37  4659.9 1472.38  4674.5 1470.78  4774.2 1466.83
  4874.0 1469.19  4909.4 1467.63  4938.4 1465.28  4952.4 1462.98  4952.9 1462.48
  4966.0 1462.98  4973.8 1464.16  5000.0 1463.41  5017.2 1465.64  5039.9 1466.13
  5125.3 1472.24  5260.5 1476.61  5436.7 1479.72  5547.0 1479.84  5577.3 1480.82
  5679.4 1480.48  5723.2 1481.62  5773.0 1481.21  5918.9 1484.08  5989.2 1484.44
#Mann=3,-1,0
  4089.4    0.05       0  4952.4    0.05       0  4966.0    0.05       0
Bank Sta=4952.4,4966
Exp/Cntr=0.3,0.1

Type RM Length L Ch R = 1,14000,500,500,500
BEGIN DESCRIPTION:
LEFT HAND CREEK 28.0
END DESCRIPTION:
XS GIS Cut Line= 3
      2748105.68     10168553.08      2748228.08     10169407.55
      2747805.65     10169903.15
#Sta/Elev= 30
  4136.8 1487.09  4454.6 1478.83  4595.8 1477.99  4601.5 1476.99  4666.5 1475.12
  4672.2 1474.16  4702.6 1472.80  4854.1 1468.87  4914.7 1465.96  4924.8 1463.89
  4975.3 1464.92  5000.0 1463.54  5006.1 1461.97  5020.3 1461.10  5033.6 1462.04
  5069.5 1460.34  5070.0 1459.84  5083.2 1460.34  5084.0 1461.16  5104.9 1461.85
  5112.4 1463.03  5168.6 1464.07  5182.8 1465.21  5246.5 1464.65  5310.2 1469.27
  5431.0 1472.57  5473.8 1474.94  5480.4 1476.05  5523.2 1477.59  5651.2 1484.65
#Mann=3,-1,0
  4136.8    0.05       0  5069.5    0.05       0  5083.2    0.05       0
Bank Sta=5069.5,5083.2
Exp/Cntr=0.3,0.1

Type RM Length L Ch R = 1,13500,500,500,500
BEGIN DESCRIPTION:
LEFT HAND CREEK 27.0
END DESCRIPTION:
XS GIS Cut Line= 3
      2748055.69     10168953.10      2747797.75     10169299.14
      2747755.68     10169703.15
#Sta/Elev= 30
  4568.4 1479.11  4696.6 1474.34  4782.1 1468.57  4825.9 1466.58  4832.2 1466.73
  4840.5 1465.89  4890.6 1463.66  4917.7 1461.74  4976.1 1460.17  4982.3 1459.56
  4992.5 1457.72  4993.0 1457.22  5005.8 1457.22  5006.3 1457.72  5024.1 1457.78
  5044.2 1460.65  5068.8 1461.36  5074.4 1462.54  5094.5 1463.48  5114.6 1463.67
  5134.7 1464.56  5185.0 1467.71  5225.2 1469.29  5315.7 1475.91  5335.8 1477.93
  5345.8 1479.34  5359.4 1479.66  5365.9 1480.46  5386.0 1480.41  5406.2 1481.13
#Mann=3,-1,0
  4568.4    0.05       0  4992.5    0.05       0  5006.3    0.05       0
Bank Sta=4992.5,5006.3
Exp/Cntr=0.3,0.1

Type RM Length L Ch R = 1,13000,500,500,500
BEGIN DESCRIPTION:
LEFT HAND CREEK 26.0
END DESCRIPTION:
XS GIS Cut Line= 3
      2747555.70     10168853.08      2747321.25     10169209.00
      2747555.70     10169603.14
#Sta/Elev= 30
  4573.8 1471.97  4632.6 1469.19  4681.6 1470.22  4695.8 1470.00  4704.9 1468.19
  4710.9 1469.35  4725.9 1466.65  4762.1 1465.21  4789.4 1461.62  4840.3 1461.56
  4891.6 1458.90  4906.6 1459.67  4992.6 1451.34  4993.1 1450.84  5006.4 1451.34
  5020.3 1453.25  5051.3 1451.76  5063.2 1453.76  5086.2 1454.07  5109.5 1456.26
  5115.8 1458.55  5174.2 1464.11  5195.6 1464.50  5211.2 1467.56  5232.6 1469.58
  5296.9 1469.67  5349.5 1472.65  5370.9 1471.39  5429.4 1473.45  5458.6 1476.10
#Mann=3,-1,0
  4573.8    0.05       0  4992.6    0.05       0  5006.4    0.05       0
Bank Sta=4992.6,5006.4
Exp/Cntr=0.3,0.1

Type RM Length L Ch R = 1,12500,500,500,500
BEGIN DESCRIPTION:
LEFT HAND CREEK 25.0
END DESCRIPTION:
XS GIS Cut Line= 3
      2746355.66     10169003.10      2746874.65     10169338.80
      2747255.69     10169753.12
#Sta/Elev= 30
  4381.9 1465.65  4404.7 1465.97  4431.7 1464.37  4477.2 1463.33  4512.9 1463.56
  4525.4 1461.75  4620.1 1460.78  4715.4 1457.63  4786.9 1454.13  4809.7 1452.09
  4815.6 1450.14  4836.7 1447.44  4867.1 1446.78  4903.3 1448.25  4924.5 1447.60
  4930.4 1446.42  4960.7 1446.08  4966.7 1445.13  4975.9 1445.73  4981.8 1444.63
  5011.1 1444.12  5011.6 1443.62  5025.2 1444.12  5060.2 1448.94  5095.9 1449.27
  5131.0 1451.15  5265.4 1455.26  5357.9 1459.98  5364.7 1459.28  5562.9 1466.17
#Mann=3,-1,0
  4381.9    0.05       0  5011.1    0.05       0  5025.2    0.05       0
Bank Sta=5011.1,5025.2
Exp/Cntr=0.3,0.1

Type RM Length L Ch R = 1,12000,500,500,500
BEGIN DESCRIPTION:
LEFT HAND CREEK 24.0
END DESCRIPTION:
XS GIS Cut Line= 3
      2746095.75     10169453.59      2746511.66     10169614.34
      2747081.27     10169856.12
#Sta/Elev= 30
  4554.1 1452.01  4677.5 1455.26  4779.2 1454.40  4895.6 1449.25  4901.0 1448.31
  4907.8 1448.83  4925.6 1447.36  4930.9 1446.19  4940.0 1446.36  4972.1 1441.99
  5008.1 1439.47  5008.6 1438.97  5022.3 1439.47  5038.8 1440.52  5057.0 1444.34
  5091.6 1445.72  5109.8 1448.39  5145.6 1450.65  5168.0 1450.43  5186.2 1451.56
  5244.4 1452.53  5286.3 1454.28  5291.7 1453.74  5339.0 1454.65  5420.9 1454.35
  5444.5 1455.29  5497.3 1455.50  5544.6 1457.55  5550.0 1456.97  5618.8 1458.20
#Mann=3,-1,0
  4554.1    0.05       0  5008.1    0.05       0  5022.3    0.05       0
Bank Sta=5008.1,5022.3
Exp/Cntr=0.3,0.1

Type RM Length L Ch R = 1,11500,500,500,500
BEGIN DESCRIPTION:
LEFT HAND CREEK 23.0
END DESCRIPTION:
XS GIS Cut Line= 3
      2746206.83     10170057.76      2746621.95     10170092.83
      2747122.08     10170127.11
#Sta/Elev= 30
  4583.4 1453.19  4587.4 1451.44  4602.3 1450.82  4612.4 1449.21  4622.4 1448.66
  4672.6 1448.08  4783.0 1442.12  4813.1 1442.91  4863.2 1440.90  4883.3 1439.39
  4893.4 1440.39  4913.4 1439.49  4946.3 1439.76  4953.6 1438.14  4966.5 1436.80
  4967.0 1436.30  4980.7 1436.80  5013.8 1438.00  5023.8 1439.92  5073.1 1442.14
  5124.0 1442.62  5144.1 1444.12  5164.1 1444.48  5284.4 1446.49  5304.4 1445.97
  5369.7 1446.99  5444.8 1446.32  5474.8 1445.67  5484.9 1444.71  5501.3 1445.82
#Mann=3,-1,0
  4583.4    0.05       0  4966.5    0.05       0  4980.7    0.05       0
Bank Sta=4966.5,4980.7
Exp/Cntr=0.3,0.1

Type RM Length L Ch R = 1,11000,500,500,500
BEGIN DESCRIPTION:
LEFT HAND CREEK 22.0
END DESCRIPTION:
XS GIS Cut Line= 3
      2746305.70     10170203.13      2746657.62     10170576.39
      2747055.73     10170503.10
#Sta/Elev= 30
  4487.0 1447.51  4522.4 1441.47  4571.7 1430.11  4593.2 1429.46  4607.3 1430.81
  4614.2 1432.91  4621.5 1431.67  4635.7 1432.11  4656.7 1434.35  4699.2 1433.49
  4776.9 1429.88  4812.5 1426.55  4883.3 1423.82  4918.5 1419.89  4939.9 1422.81
  4974.9 1417.39  4975.4 1416.89  4989.1 1417.39  5044.7 1422.61  5097.8 1424.16
  5120.0 1423.34  5214.0 1427.67  5252.2 1430.90  5292.9 1440.43  5320.1 1449.75
  5343.7 1451.87  5364.1 1457.50  5378.2 1458.31  5384.4 1460.13  5404.8 1459.95
#Mann=3,-1,0
  4487.0    0.05       0  4974.9    0.05       0  4989.1    0.05       0
Bank Sta=4974.9,4989.1
Exp/Cntr=0.3,0.1

Type RM Length L Ch R = 1,10500,500,500,500
BEGIN DESCRIPTION:
LEFT HAND CREEK 21.0
END DESCRIPTION:
XS GIS Cut Line= 3
      2746061.02     10170224.40      2746217.22     10170669.06
      2746206.91     10171160.05
#Sta/Elev= 30
  4528.7 1440.15  4555.8 1436.06  4580.3 1434.53  4648.8 1432.72  4686.3 1430.16
  4760.5 1427.90  4834.7 1423.49  4860.4 1422.92  4917.1 1419.96  4922.4 1420.40
  4940.7 1418.74  4948.1 1417.29  4953.4 1418.31  4991.9 1414.97  4992.4 1414.47
  5007.0 1414.97  5024.1 1416.02  5044.1 1419.13  5074.1 1417.94  5104.1 1418.86
  5114.1 1420.35  5134.1 1419.06  5154.1 1419.37  5184.1 1417.57  5244.1 1418.67
  5324.1 1423.82  5384.1 1426.48  5414.1 1424.83  5463.0 1425.63  5491.1 1426.59
#Mann=4,-1,0
  4528.7    0.05       0  4991.9    0.05       0  5007.0    0.05       0
  5463.0    0.12       0
Bank Sta=4991.9,5007
Exp/Cntr=0.3,0.1

Type RM Length L Ch R = 1,10000,500,500,500
BEGIN DESCRIPTION:
LEFT HAND CREEK 20.0
END DESCRIPTION:
XS GIS Cut Line= 3
      2745894.36     10170280.03      2745789.03     10170722.26
      2745700.31     10171014.81
#Sta/Elev= 30
  4545.4 1424.23  4569.1 1424.23  4589.7 1425.21  4652.0 1422.54  4795.3 1418.44
  4815.5 1419.06  4857.0 1417.84  4904.9 1414.83  4939.2 1414.18  4947.0 1413.59
  4962.4 1410.14  4962.9 1409.64  4977.6 1410.14  4994.3 1410.52  4997.9 1411.72
  5011.3 1412.71  5027.9 1412.54  5066.0 1414.89  5105.4 1420.22  5115.8 1420.72
  5131.8 1426.35  5137.0 1426.73  5157.6 1427.27  5164.7 1425.95  5169.9 1426.03
  5178.5 1424.20  5209.9 1425.71  5230.5 1425.60  5235.8 1426.33  5305.7 1426.66
#Mann=3,-1,0
  4545.4    0.05       0  4962.4    0.03       0  4977.6    0.05       0
Bank Sta=4962.4,4977.6
Exp/Cntr=0.3,0.1

Type RM Length L Ch R = 1,9500,500,500,500
BEGIN DESCRIPTION:
LEFT HAND CREEK 19.0
END DESCRIPTION:
XS GIS Cut Line= 3
      2745463.81     10170064.75      2745409.67     10170531.82
      2745505.69     10170803.13
#Sta/Elev= 30
  4529.8 1424.10  4568.4 1421.12  4598.6 1422.79  4727.5 1421.00  4870.4 1412.56
  4890.6 1410.13  4905.0 1412.06  4920.8 1412.35  4990.5 1407.27  4991.0 1406.77
  5005.7 1407.27  5054.4 1409.57  5061.4 1408.35  5066.7 1410.48  5086.2 1408.43
  5097.6 1411.76  5107.4 1413.16  5117.8 1413.19  5171.1 1420.35  5179.6 1420.35
  5184.9 1423.59  5192.3 1424.76  5210.5 1424.87  5215.8 1427.82  5234.7 1424.44
  5241.4 1424.91  5246.7 1429.60  5272.3 1428.19  5277.6 1430.52  5287.8 1430.41
#Mann=3,-1,0
  4529.8    0.05       0  4990.5    0.05       0  5005.7    0.05       0
Bank Sta=4990.5,5005.7
Exp/Cntr=0.3,0.1

Type RM Length L Ch R = 1,9000,500,500,500
BEGIN DESCRIPTION:
LEFT HAND CREEK 18.0
END DESCRIPTION:
XS GIS Cut Line= 3
      2744805.70     10170603.13      2745134.36     10170940.92
      2745405.64     10170903.12
#Sta/Elev= 30
  4528.7 1420.73  4535.8 1419.49  4600.5 1416.71  4634.8 1413.86  4652.0 1414.29
  4712.0 1410.28  4769.1 1409.50  4832.8 1407.03  4875.3 1402.30  4890.3 1401.98
  4917.7 1401.10  4924.7 1401.91  4931.8 1400.53  4938.8 1401.13  4973.1 1398.26
  4973.6 1397.76  4989.4 1398.26  4998.0 1399.88  5023.5 1399.45  5072.0 1402.47
  5095.0 1402.65  5132.6 1408.43  5161.6 1409.96  5173.0 1409.44  5183.1 1410.93
  5203.3 1419.24  5213.4 1419.46  5243.7 1428.19  5263.8 1425.87  5273.9 1425.85
#Mann=7,-1,0
  4528.7    0.05       0  4600.5    0.12       0  4652.0    0.05       0
  4712.0    0.12       0  4890.3    0.05       0  4973.1    0.05       0
  4989.4    0.05       0
Bank Sta=4973.1,4989.4
Exp/Cntr=0.3,0.1

Type RM Length L Ch R = 1,8500,500,500,500
BEGIN DESCRIPTION:
LEFT HAND CREEK 17.0
END DESCRIPTION:
XS GIS Cut Line= 3
      2744305.66     10170803.09      2744797.54     10171302.97
      2745755.66     10171503.11
#Sta/Elev= 30
  4298.7 1414.64  4461.4 1411.56  4744.3 1401.84  4829.1 1400.63  4921.0 1401.64
  4942.3 1398.77  5010.4 1394.52  5010.9 1394.02  5026.7 1394.52  5110.5 1399.07
  5151.3 1396.07  5182.0 1400.87  5233.1 1403.77  5345.4 1404.15  5478.2 1409.76
  5600.8 1412.15  5659.0 1416.81  5723.4 1419.61  5733.6 1421.66  5753.9 1429.78
  5759.0 1428.85  5768.0 1432.53  5784.7 1435.90  5815.4 1437.34  5835.7 1441.67
  5853.8 1444.94  5858.9 1443.82  5867.9 1446.33  5938.0 1453.10  5978.8 1454.50
#Mann=6,-1,0
  4298.7    0.05       0  5010.4    0.05       0  5026.7    0.05       0
  5768.0    0.12       0  5835.7    0.05       0  5867.9    0.12       0
Bank Sta=5010.4,5026.7
Exp/Cntr=0.3,0.1

Type RM Length L Ch R = 1,8000,500,500,500
BEGIN DESCRIPTION:
LEFT HAND CREEK 16.0
END DESCRIPTION:
XS GIS Cut Line= 3
      2744305.69     10170953.14      2744343.17     10171431.07
      2745005.70     10171953.12
#Sta/Elev= 30
  4520.6 1412.49  4714.3 1405.59  4831.5 1399.24  4941.9 1399.19  4961.9 1393.52
  4964.4 1391.19  4964.9 1390.69  4980.9 1391.19  4999.6 1391.26  5025.8 1392.26
  5039.4 1391.82  5066.9 1393.61  5089.1 1392.88  5109.9 1394.47  5124.3 1393.61
  5181.4 1397.49  5194.8 1399.67  5238.2 1403.02  5295.9 1405.08  5308.8 1406.83
  5366.4 1404.63  5395.3 1406.20  5430.6 1404.87  5523.6 1406.01  5579.7 1407.88
  5587.8 1409.92  5614.9 1409.03  5651.9 1411.36  5786.6 1411.56  5843.5 1414.19
#Mann=5,-1,0
  4520.6    0.05       0  4964.4    0.07       0  4980.9    0.05       0
  4999.6    0.12       0  5025.8    0.05       0
Bank Sta=4964.4,4980.9
Exp/Cntr=0.3,0.1
