--- MARSCHALL BRANCH.prj (project) ---

Proj Title=MARSCHALL BRANCH Base Level Engineering
Current Plan=p01
Default Exp/Contr=0.3,0.1
English Units
Geom File=g01
Flow File=f01
Plan File=p01
Y Axis Title=Elevation
X Axis Title(PF)=Main Channel Distance
X Axis Title(XS)=Station
BEGIN DESCRIPTION:
MARSCHALL BRANCH
END DESCRIPTION:
DSS Export Rating Curves= 0
DSS Export Rating Curve Sorted= 0
DSS Export Volume Flow Curves= 0
DXF OffsetX= 0
DXF OffsetY= 0
DXF ScaleX= 1
DXF ScaleY= 10

--- MARSCHALL BRANCH.p01 (plan) ---

Plan Title=Multiple Run
Short Identifier=Multiple
Geom File=g01
Flow File=f01
Subcritical Flow
K Sum by GR= 0
Std Step Tol= 0.01
Critical Tol= 0.01
Num of Std Step Trials= 20
Max Error Tol= 0.3
Flow Tol Ratio= 0.001
Split Flow NTrial= 30
Split Flow Tol= 0.02
Split Flow Ratio= 0.02
Log Output Level= 0
Friction Slope Method= 1
Unsteady Friction Slope Method= 2
Unsteady Bridges Friction Slope Method= 1
Parabolic Critical Depth
Global Vel Dist=  1 , 1 , 1
Global Log Level= 0
CheckData=True
Encroach Param= -1, 0, 0, 0
BEGIN DESCRIPTION:
Multiple Run
END DESCRIPTION:

--- MARSCHALL BRANCH.f01 (steady flow) ---

Flow Title=Multiple
Program Version=4.10
Number of Profiles= 7
Profile Names=10-year,25-year,50-year,1pct_min,100-year,1pct_plu,500-year
River Rch & RM=MARSCHALL BRANCH,Reach-1         ,21826
    6313   12105   20541   13036   30017   69122   40720
River Rch & RM=MARSCHALL BRANCH,Reach-1         ,17500
    8618   16492   27643   17340   40202   93209   53957
River Rch & RM=MARSCHALL BRANCH,Reach-1         ,9500
   10141   19329   31884   24517   46134   86809   61435
River Rch & RM=MARSCHALL BRANCH,Reach-1         ,6000
   10321   19669   32404   24911   46879   88221   62401
River Rch & RM=MARSCHALL BRANCH,Reach-1         ,3500
   15155   28536   45514   34078   65055  124191   85258
River Rch & RM=MARSCHALL BRANCH,Reach-1         ,578
   15278   28766   45885   34340   65585  125260   85952
Boundary for River Rch & Prof#=MARSCHALL BRANCH,Reach-1         , 1
Up Type= 0
Dn Type= 3
Dn Slope=0.001
Boundary for River Rch & Prof#=MARSCHALL BRANCH,Reach-1         , 2
Up Type= 0
Dn Type= 3
Dn Slope=0.001
Boundary for River Rch & Prof#=MARSCHALL BRANCH,Reach-1         , 3
Up Type= 0
Dn Type= 3
Dn Slope=0.001
Boundary for River Rch & Prof#=MARSCHALL BRANCH,Reach-1         , 4
Up Type= 0
Dn Type= 3
Dn Slope=0.001
Boundary for River Rch & Prof#=MARSCHALL BRANCH,Reach-1         , 5
Up Type= 0
Dn Type= 3
Dn Slope=0.001
Boundary for River Rch & Prof#=MARSCHALL BRANCH,Reach-1         , 6
Up Type= 0
Dn Type= 3
Dn Slope=0.001
Boundary for River Rch & Prof#=MARSCHALL BRANCH,Reach-1         , 7
Up Type= 0
Dn Type= 3
Dn Slope=0.001
DSS Import GetInterval= 0
DSS Import GetPeak= 0
DSS Import FillOption= 0

--- MARSCHALL BRANCH.g01 (geometry) ---

Geom Title=Existing Conditions
Program Version=4.10

River Reach=MARSCHALL BRANCH,Reach-1
Reach XY= 30
        2727650.       10166517.        2727801.       10167567.
        2727726.       10167751.      2728204.25       10168511.
       2728360.5       10168945.      2728254.25       10169264.
        2727726.       10169548.        2727698.       10169848.
        2727871.       10170100.      2728508.25       10170194.
      2729004.25       10170705.        2729351.       10171289.
      2729194.75       10171711.       2729285.5       10172026.
      2729157.25       10173073.       2729252.5       10173202.
       2729913.5       10173464.      2730244.75       10173964.
        2730726.       10175286.      2730677.25       10176110.
       2730835.5       10176411.        2731526.       10177151.
        2731398.       10178661.      2731632.25       10179142.
       2732937.5       10180135.      2733388.25       10180308.
        2733991.       10180977.      2734634.75       10181226.
        2735094.       10181195.      2737129.75       10181780.

Type RM Length L Ch R = 1 ,21826   ,500,500,500
BEGIN DESCRIPTION:
MARSCHALL BRANCH 43.0
END DESCRIPTION:
XS GIS Cut Line= 3
      2727154.04     10166726.63      2727475.65     10166592.51
      2728138.41     10166339.91
#Sta/Elev= 30
       0 1482.44   208.5 1476.26   256.2 1474.22   303.8 1470.97   362.7 1468.48
   380.6 1466.52   392.8 1466.38     402 1465.34   434.1 1463.94   447.6 1462.95
   455.5 1461.17   477.7 1461.15   527.2 1459.15   532.5 1460.37   562.6    1464
   573.2 1465.36   642.2 1467.55   648.1 1469.27   702.4 1470.57   751.9 1473.18
   757.2 1472.64     798 1474.54   830.1 1476.14   836.8 1477.65   883.6 1478.63
   921.7 1480.38   951.8 1480.43   976.5 1482.16  1006.6 1482.73  1057.7 1485.54
#Mann= 3 , 0 , 0
       0     .05       0   434.1     .03       0   562.6     .05       0
Bank Sta=434.1,562.6
XS Rating Curve= 0 ,0
Exp/Cntr=0.3,0.1

Type RM Length L Ch R = 1 ,21000   ,500,500,500
BEGIN DESCRIPTION:
MARSCHALL BRANCH 42.0
END DESCRIPTION:
XS GIS Cut Line= 3
      2727255.72      10167553.1      2727773.75     10167324.58
      2728255.66     10166903.13
#Sta/Elev= 30
  4433.8 1483.71  4448.2 1483.42  4494.8 1478.55  4541.4 1477.13  4616.9  1471.4
  4814.3 1463.76  4918.5 1462.74  4947.5 1459.37  4970.6 1460.12    4994 1457.48
  4998.3 1455.36  4999.1 1454.86  5034.1 1455.36  5080.7 1459.76  5101.6 1459.49
  5122.5  1461.7  5144.3 1461.79  5150.9 1463.55  5158.5 1461.63    5187 1462.37
  5279.1 1467.21  5314.2 1467.17  5342.7  1470.2  5349.3 1469.16  5363.6 1469.73
  5385.4 1471.92  5413.9 1472.21  5420.5 1471.23  5569.5 1478.65  5640.2 1480.35
#Mann= 3 ,-1 , 0
  4433.8     .05       0  4998.3     .05       0  5034.1     .05       0
Bank Sta=4998.3,5034.1
XS Rating Curve= 0 ,0
Exp/Cntr=0.3,0.1

Type RM Length L Ch R = 1 ,20500   ,500,500,500
BEGIN DESCRIPTION:
MARSCHALL BRANCH 41.0
END DESCRIPTION:
XS GIS Cut Line= 3
       2727405.7      10167903.1      2727741.74     10167791.75
      2728555.91     10167498.13
#Sta/Elev= 30
    4646 1474.21  4825.6 1466.99    4852 1468.61  4877.7 1465.94  4883.7 1467.73
    4889 1466.56  4898.8  1467.9  4920.7 1462.45  4972.6 1459.23  4978.8  1457.2
  4984.1 1457.31  4992.2 1450.35    4993 1449.85    5028 1450.35  5035.5 1452.96
  5066.2 1454.87  5071.5 1454.25  5096.9 1456.68  5102.2  1455.8  5132.9 1456.11
  5142.4 1457.41  5158.2 1457.42  5227.4 1454.57    5245 1459.11  5291.2 1460.25
  5312.5 1462.56  5344.4 1463.76  5597.2 1467.54    5776  1474.4  5865.5  1475.8
#Mann= 3 ,-1 , 0
    4646     .05       0  4992.2     .05       0    5028     .05       0
Bank Sta=4992.2,5028
XS Rating Curve= 0 ,0
Exp/Cntr=0.3,0.1

Type RM Length L Ch R = 1 ,20000   ,500,500,500
BEGIN DESCRIPTION:
MARSCHALL BRANCH 40.0
END DESCRIPTION:
XS GIS Cut Line= 3
      2727375.38     10168426.94      2727993.71     10168220.44
      2728790.29     10167749.86
#Sta/Elev= 30
  4348.1 1466.08  4453.9 1467.42  4559.3 1465.67    4565  1466.5  4622.5 1466.08
  4659.8 1467.59  4738.5 1467.92  4791.4 1467.88  4849.4 1465.92  4875.6 1466.67
    4881 1465.01  4886.2 1465.95  4912.6 1460.64  4938.8 1457.52  4944.2 1456.06
  4959.9 1455.15    4981 1451.26  4988.4 1447.11  4989.2 1446.61  5024.3 1447.11
  5043.4  1450.6  5086.3 1455.07  5095.2 1454.12  5163.3 1456.73  5234.6 1461.83
    5313 1463.68  5453.1 1465.23  5735.9 1471.74  5831.5 1471.72  5925.2  1469.9
#Mann= 5 ,-1 , 0
  4348.1     .05       0  4988.4     .05       0  5024.3     .05       0
  5163.3     .12       0    5313     .05       0
Bank Sta=4988.4,5024.3
XS Rating Curve= 0 ,0
Exp/Cntr=0.3,0.1

Type RM Length L Ch R = 1 ,19500   ,500,500,500
BEGIN DESCRIPTION:
MARSCHALL BRANCH 39.0
END DESCRIPTION:
XS GIS Cut Line= 3
      2727436.12     10168617.91      2728257.39     10168641.23
      2729406.58     10168643.95
#Sta/Elev= 30
  4178.4 1459.21    4248 1458.07    4268 1459.21    4288 1457.94  4418.1 1456.77
  4508.1 1458.37  4648.2  1457.1  4768.2  1460.2  4886.6 1455.71  4891.6 1456.27
  4968.3  1450.7  4996.6 1446.15  5010.3 1446.01  5011.2 1445.51  5046.2 1446.01
  5058.3  1448.7  5078.3 1450.61  5168.3 1452.25  5198.3 1454.78  5238.3 1455.19
  5248.3 1456.23  5408.3 1457.32  5548.3 1456.05  5568.3    1455  5598.3 1455.64
  5628.3 1458.16  5658.3 1458.04  5808.3  1463.9  5888.3 1468.68  6149.2 1471.84
#Mann= 3 ,-1 , 0
  4178.4     .05       0  5010.3     .05       0  5046.2     .05       0
Bank Sta=5010.3,5046.2
XS Rating Curve= 0 ,0
Exp/Cntr=0.3,0.1

Type RM Length L Ch R = 1 ,19000   ,500,500,500
BEGIN DESCRIPTION:
MARSCHALL BRANCH 38.0
END DESCRIPTION:
XS GIS Cut Line= 3
      2727332.02      10168982.5      2728333.18     10169117.31
      2728755.73      10169053.1
#Sta/Elev= 30
  3989.8 1465.03    4276 1454.29  4336.6 1454.32  4366.8 1455.97  4376.9  1457.7
    4387 1457.49  4417.3 1454.28  4447.6  1453.7    4560 1446.59  4627.7 1451.04
  4632.8 1450.14  4705.6 1451.68  4710.6 1450.35  4778.4 1450.59    4831 1447.23
  4861.3 1447.85  4891.5 1444.52    4929 1446.09  4962.2 1443.59  4994.6 1442.89
  4995.4 1442.39  5030.7 1442.89  5032.9 1445.09  5064.8 1445.91  5073.3 1444.83
  5093.6 1446.09  5103.7 1447.02  5123.3 1451.37  5174.5    1451  5427.4 1463.88
#Mann= 3 ,-1 , 0
  3989.8     .05       0  4994.6     .03       0  5030.7     .05       0
Bank Sta=4994.6,5030.7
XS Rating Curve= 0 ,0
Exp/Cntr=0.3,0.1

Type RM Length L Ch R = 1 ,18500   ,500,500,500
BEGIN DESCRIPTION:
MARSCHALL BRANCH 37.0
END DESCRIPTION:
XS GIS Cut Line= 3
      2727455.72     10169353.12      2727966.01     10169422.65
      2728605.68     10169453.11
#Sta/Elev= 30
    4485 1460.09  4505.1 1457.78  4545.5 1458.15  4565.7 1455.14  4593.5 1447.93
  4598.5 1448.64  4616.2 1444.91  4665.9    1443  4670.9 1444.84  4676.7 1442.86
  4696.9 1441.07  4727.2 1442.01  4815.6 1440.78  4838.2 1437.09    4888 1439.82
  4979.5 1436.26  5039.7 1438.99  5089.8 1437.26  5091.8 1435.59  5092.6 1435.09
  5127.9 1435.59  5219.9 1440.42    5250 1449.29    5280 1447.44    5300 1442.34
    5310 1444.68  5330.1 1444.04  5360.1  1452.4  5410.1 1450.52  5640.4 1460.05
#Mann= 3 ,-1 , 0
    4485     .05       0  5091.8     .05       0  5127.9     .05       0
Bank Sta=5091.8,5127.9
XS Rating Curve= 0 ,0
Exp/Cntr=0.3,0.1

Type RM Length L Ch R = 1 ,18000   ,500,500,500
BEGIN DESCRIPTION:
MARSCHALL BRANCH 36.0
END DESCRIPTION:
XS GIS Cut Line= 3
      2727505.64      10169703.1       2727687.2     10169764.64
      2728655.71     10169503.11
#Sta/Elev= 30
  4808.3 1461.94  4861.1 1458.44  4881.6 1452.07  4886.9 1453.66  4892.8 1447.67
    4913 1442.99  4918.3 1443.53  4935.1 1439.46  4949.7 1439.41  4966.7 1435.18
  4981.1 1434.85  5008.8 1427.42  5029.9 1428.26  5032.2 1426.36    5033 1425.86
  5068.3 1426.36  5070.9 1428.39  5226.3 1430.35  5253.7 1434.48  5309.2    1434
  5319.5  1435.9  5333.5 1434.17  5454.2 1440.33  5487.9 1440.35  5527.8 1437.51
  5602.4 1443.84  5642.3 1449.19  5702.8 1448.59  5911.2 1459.07  6003.2  1461.2
#Mann= 3 ,-1 , 0
  4808.3     .05       0  5032.2     .05       0  5068.3     .05       0
Bank Sta=5032.2,5068.3
XS Rating Curve= 0 ,0
Exp/Cntr=0.3,0.1

Type RM Length L Ch R = 1 ,17500   ,500,500,500
BEGIN DESCRIPTION:
MARSCHALL BRANCH 35.0
END DESCRIPTION:
XS GIS Cut Line= 3
      2727605.69     10170353.11      2727979.92     10170104.11
      2728355.69     10169753.11
#Sta/Elev= 30
  4550.5 1443.43  4586.5 1443.61  4651.2 1438.73  4744.4 1436.41  4759.4 1435.24
  4766.7 1433.39  4831.5 1430.43  4867.6 1430.62  4882.6 1429.02  4888.6 1427.04
  4897.7 1426.64  4903.7 1424.32  4924.7 1422.28    5012 1417.85    5013 1417.35
  5054.5 1417.85  5068.4 1423.29  5082.6 1425.31  5089.9  1424.4  5103.7  1425.7
  5125.1 1423.45  5153.4 1428.72  5174.4 1430.01  5195.9 1429.95  5252.6 1433.88
  5393.8 1437.32  5422.1 1440.83  5464.6 1442.03  5486.1  1444.5  5514.2 1444.85
#Mann= 3 ,-1 , 0
  4550.5     .05       0    5012     .05       0  5054.5     .05       0
Bank Sta=5012,5054.5
XS Rating Curve= 0 ,0
Exp/Cntr=0.3,0.1

Type RM Length L Ch R = 1 ,17000   ,500,500,500
BEGIN DESCRIPTION:
MARSCHALL BRANCH 34.0
END DESCRIPTION:
XS GIS Cut Line= 3
      2727960.63     10170745.26      2728469.38     10170163.54
      2728705.67     10170103.11
#Sta/Elev= 30
  4227.2 1443.39  4260.5 1443.79  4473.1 1438.06  4550.9 1433.54  4579.4 1430.69
  4699.9 1425.09    4735 1426.83  4749.3  1426.2    4792 1430.17  4834.7 1425.47
  4905.9  1424.5  4926.8 1422.89    4941 1419.84  4969.5 1416.39  4995.5 1415.42
  4996.5 1414.92    5038 1415.42  5047.8 1422.17  5057.6 1423.31  5062.8 1425.46
  5078.8 1426.94  5103.6 1435.48  5109.7 1438.57    5120 1440.37  5139.3 1442.23
  5144.4 1443.78  5180.1 1442.14  5202.6 1445.39  5220.9 1451.14  5243.9 1450.54
#Mann= 3 ,-1 , 0
  4227.2     .05       0  4995.5     .05       0    5038     .05       0
Bank Sta=4995.5,5038
XS Rating Curve= 0 ,0
Exp/Cntr=0.3,0.1

Type RM Length L Ch R = 1 ,16500   ,500,500,500
BEGIN DESCRIPTION:
MARSCHALL BRANCH 33.0
END DESCRIPTION:
XS GIS Cut Line= 3
      2728605.68     10170803.12      2728785.05     10170547.22
      2728905.66     10170353.15
#Sta/Elev= 30
  4687.5  1436.7  4694.9 1436.95    4701 1435.44  4724.1 1433.32  4730.7 1433.99
  4745.5 1432.83  4760.3 1430.01  4781.2 1430.65  4852.7 1426.58  4858.8 1425.34
  4867.5 1425.47  4873.6 1424.13  4918.1 1422.78  4968.4  1417.6  4974.4 1414.36
  4975.4 1413.86  5016.9 1414.36  5026.1 1415.23  5031.9 1414.43  5083.9 1415.81
    5099 1417.48    5111 1421.19  5126.4 1423.52  5134.4 1426.72  5141.8 1431.56
  5157.1 1430.48    5163 1428.88  5178.4 1428.91  5205.5 1434.53  5228.5 1436.44
#Mann= 3 ,-1 , 0
  4687.5     .05       0  4974.4     .05       0  5016.9     .05       0
Bank Sta=4974.4,5016.9
XS Rating Curve= 0 ,0
Exp/Cntr=0.3,0.1

Type RM Length L Ch R = 1 ,16000   ,500,500,500
BEGIN DESCRIPTION:
MARSCHALL BRANCH 32.0
END DESCRIPTION:
XS GIS Cut Line= 3
      2728655.71     10171303.09      2729130.95     10170892.72
      2729255.69     10170553.11
#Sta/Elev= 30
  4372.1 1435.65  4464.6  1429.6  4485.6 1429.51  4514.1 1427.64    4592 1425.07
  4641.4 1424.71  4684.1  1422.6  4690.8 1423.22  4811.4 1420.74  4903.6 1417.23
  4932.1 1415.76  4939.3 1411.01  4940.3 1410.51  4981.8 1411.01  5027.2 1411.75
  5032.6 1412.72  5052.4 1413.33  5095.5 1419.35  5127.4 1421.05  5143.8 1424.15
  5149.2 1423.31  5199.5 1424.56  5204.8  1425.4  5212.6 1424.68    5230 1425.88
  5244.6 1425.49  5285.6 1427.32  5308.5 1430.91  5316.1 1430.31  5361.8 1434.91
#Mann= 3 ,-1 , 0
  4372.1     .05       0  4939.3     .03       0  4981.8     .05       0
Bank Sta=4939.3,4981.8
XS Rating Curve= 0 ,0
Exp/Cntr=0.3,0.1

Type RM Length L Ch R = 1 ,15500   ,500,500,500
BEGIN DESCRIPTION:
MARSCHALL BRANCH 31.0
END DESCRIPTION:
XS GIS Cut Line= 3
      2728855.71      10171703.1      2729361.75     10171320.83
      2729605.73      10171253.1
#Sta/Elev= 30
  4365.8 1426.88  4373.1 1424.24  4393.9 1421.51  4502.1 1413.32  4508.3 1414.54
  4593.7 1414.16  4666.5 1411.19  4701.9 1412.96  4779.3  1409.1  4793.5 1411.46
  4801.8 1410.94    4808 1412.98  4837.2 1408.82  4866.3  1409.8  4872.6 1411.42
  4887.1 1409.46  4922.5 1409.54  4937.1 1406.86  4943.3 1407.74  4965.7 1405.59
  4966.7 1405.09  5008.3 1405.59  5024.8 1408.38  5066.3 1409.67  5083.4 1415.33
  5088.6 1414.64  5117.7 1425.27  5122.9 1424.62  5180.5  1435.1  5253.2 1440.21
#Mann= 3 ,-1 , 0
  4365.8     .05       0  4965.7     .05       0  5008.3     .05       0
Bank Sta=4965.7,5008.3
XS Rating Curve= 0 ,0
Exp/Cntr=0.3,0.1

Type RM Length L Ch R = 1 ,15000   ,500,500,500
BEGIN DESCRIPTION:
MARSCHALL BRANCH 30.0
END DESCRIPTION:
XS GIS Cut Line= 3
       2728855.7     10171903.11      2729210.54     10171778.46
      2729605.68     10171603.11
#Sta/Elev= 30
  4623.9 1432.98  4655.7 1431.33  4701.4 1422.71  4732.3 1420.69  4763.3 1415.51
  4782.9 1415.09    4789 1411.78  4814.7 1407.67  4824.4  1401.9  4825.4  1401.4
    4867  1401.9  4867.7 1403.67  4899.5 1403.47  4920.7 1405.68    5000 1405.65
  5016.6 1406.57  5023.8 1409.58  5029.2 1408.16  5082.2 1413.06  5151.1 1412.45
  5174.3 1415.88  5180.7 1420.41  5197.6 1424.19  5203.1 1427.45  5272.9 1428.46
  5301.6 1435.92    5312 1436.54  5371.4 1432.68  5410.4 1435.47  5432.3 1440.62
#Mann= 3 ,-1 , 0
  4623.9     .05       0  4824.4     .05       0    4867     .05       0
Bank Sta=4824.4,4867
XS Rating Curve= 0 ,0
Exp/Cntr=0.3,0.1

Type RM Length L Ch R = 1 ,14500   ,500,500,500
BEGIN DESCRIPTION:
MARSCHALL BRANCH 29.0
END DESCRIPTION:
XS GIS Cut Line= 3
      2728790.27     10172176.93      2729213.88     10172247.84
      2729597.61     10172255.06
#Sta/Elev= 30
  4570.5 1430.65  4606.4 1428.69  4626.7 1428.77  4657.1 1425.66  4700.8 1424.25
  4738.2 1424.86  4748.4 1423.01  4756.4 1419.98  4761.5  1420.4  4768.6 1418.65
    4799 1418.04  4829.5 1411.35  4882.9 1406.33  4920.7 1400.24  4922.2  1396.4
  4923.2  1395.9  4964.9  1396.4  4971.4 1399.08  4981.6 1397.73  5003.4 1397.93
  5021.8 1396.47  5051.8 1401.52  5071.8 1410.28  5121.8 1417.45  5141.8 1419.38
  5171.8 1420.25  5191.8 1418.57  5231.8  1418.8  5341.9 1423.68  5383.8 1427.98
#Mann= 3 ,-1 , 0
  4570.5     .05       0  4922.2     .05       0  4964.9     .05       0
Bank Sta=4922.2,4964.9
XS Rating Curve= 0 ,0
Exp/Cntr=0.3,0.1

Type RM Length L Ch R = 1 ,14000   ,500,500,500
BEGIN DESCRIPTION:
MARSCHALL BRANCH 28.0
END DESCRIPTION:
XS GIS Cut Line= 3
      2728642.74     10172793.26      2729176.71     10172744.39
      2729632.33     10172697.77
#Sta/Elev= 30
  4463.8 1419.22  4547.1  1414.2  4607.3 1412.15  4717.8 1405.32  4788.1 1401.73
  4808.2 1401.51  4851.4 1397.18  4868.4 1393.67  4908.6 1394.46  4917.4 1393.52
  4918.4 1393.02  4960.1 1393.52  4961.5  1394.6    5000 1394.25  5019.1 1395.06
  5049.2 1397.64  5069.3 1401.18  5089.4 1400.79  5119.6 1402.68  5139.7 1402.09
  5230.2 1405.42  5250.3 1408.05  5256.7 1410.32  5261.8 1409.19  5280.4 1412.16
  5320.6 1414.34  5340.7 1416.77    5391 1418.29  5401.1 1419.52    5458 1419.83
#Mann= 3 ,-1 , 0
  4463.8     .05       0  4917.4     .05       0  4960.1     .05       0
Bank Sta=4917.4,4960.1
XS Rating Curve= 0 ,0
Exp/Cntr=0.3,0.1

Type RM Length L Ch R = 1 ,13500   ,500,500,500
BEGIN DESCRIPTION:
MARSCHALL BRANCH 27.0
END DESCRIPTION:
XS GIS Cut Line= 3
      2728905.72     10173453.09      2729256.04     10173203.74
      2729355.68     10173003.12
#Sta/Elev= 30
    4570 1417.18  4583.5 1415.07  4633.9 1410.95  4642.5 1411.42  4648.7 1410.11
  4699.1 1405.86  4705.2 1404.78  4778.6 1401.08  4820.8 1397.56  4871.2 1391.33
    4886 1391.29  4906.9 1388.97  4921.6  1389.7  4963.4 1388.61    4972 1387.44
  4975.4 1384.24  4976.4 1383.74  5017.1 1383.74  5018.1 1384.24  5030.8 1386.16
  5036.4 1385.51  5053.2 1387.02  5067.7 1391.08  5081.2 1393.77    5126 1399.72
  5142.8 1399.18  5179.4 1403.02    5210 1403.68  5215.6 1404.84    5224 1404.55
#Mann= 3 ,-1 , 0
    4570     .05       0  4975.4     .05       0  5018.1     .05       0
Bank Sta=4975.4,5018.1
XS Rating Curve= 0 ,0
Exp/Cntr=0.3,0.1

Type RM Length L Ch R = 1 ,13000   ,500,500,500
BEGIN DESCRIPTION:
MARSCHALL BRANCH 26.0
END DESCRIPTION:
XS GIS Cut Line= 3
      2729505.66     10173753.15      2729729.22     10173358.81
       2729655.7     10173153.15
#Sta/Elev= 30
  4546.7 1404.06  4560.4 1403.51  4576.3 1406.42  4582.1 1404.28  4592.2 1405.03
  4619.6 1400.24  4635.5 1401.26  4641.2 1398.02  4650.2  1397.3  4662.9 1392.99
    4673 1392.73  4678.7 1390.01  4743.6 1384.18  4802.8 1381.06  4840.3 1385.34
  4846.1 1382.23  4856.2 1382.15  4877.8 1376.29  4899.5 1378.44  4949.1 1377.04
  4964.4 1378.71  4972.1 1376.36  4973.3  1374.2  4974.3  1373.7    5016  1374.2
  5069.8 1381.59    5116 1383.24  5146.8 1389.41  5208.4 1393.88  5218.4 1396.42
#Mann= 3 ,-1 , 0
  4546.7     .05       0  4973.3     .05       0    5016     .05       0
Bank Sta=4973.3,5016
XS Rating Curve= 0 ,0
Exp/Cntr=0.3,0.1

Type RM Length L Ch R = 1 ,12500   ,500,500,500
BEGIN DESCRIPTION:
MARSCHALL BRANCH 25.0
END DESCRIPTION:
XS GIS Cut Line= 3
      2729614.97     10173904.36      2730106.11     10173675.84
      2730505.64     10173603.12
#Sta/Elev= 30
  4458.3  1392.7  4548.5 1387.62  4594.3 1383.74  4754.5 1375.49    4790 1375.91
  4800.2 1374.09    4812 1373.89  4823.1 1375.21  4834.1 1375.03  4874.4 1372.53
  4889.2    1375  4920.2 1376.53  4955.4 1374.43  4994.3 1369.95  5002.3 1370.71
  5008.7 1369.58  5009.7 1369.08  5051.5 1369.58  5060.6 1372.15    5091 1373.75
  5150.9 1371.31  5182.5 1372.59  5202.9 1371.52  5253.7 1379.12  5267.7 1383.69
  5284.2 1392.75  5294.3 1395.62  5326.1 1394.72  5345.2 1392.55  5406.1 1392.27
#Mann= 3 ,-1 , 0
  4458.3     .05       0  5008.7     .05       0  5051.5     .05       0
Bank Sta=5008.7,5051.5
XS Rating Curve= 0 ,0
Exp/Cntr=0.3,0.1

Type RM Length L Ch R = 1 ,12000   ,500,500,500
BEGIN DESCRIPTION:
MARSCHALL BRANCH 24.0
END DESCRIPTION:
XS GIS Cut Line= 3
      2729745.13     10174199.51      2730262.06     10174139.51
      2730795.52     10174008.53
#Sta/Elev= 30
  4479.6 1387.56  4560.7  1385.7  4590.9 1383.72  4651.3 1382.51  4681.5 1380.34
  4741.9 1378.56  4843.1 1371.24  4892.9 1369.36  4921.7 1364.49  4943.2 1365.18
  4963.4 1364.04  5043.8 1363.73  5055.2 1364.55    5069 1362.96    5070 1362.46
    5112 1362.96    5117 1365.59  5132.1 1365.85  5158.2 1369.07  5173.6 1369.52
  5189.1 1371.81  5209.7    1373  5240.6 1380.28  5261.9 1378.28  5271.5 1378.48
  5298.3 1381.05  5303.5 1380.47  5386.6 1383.54  5456.8 1384.38  5549.3 1388.97
#Mann= 3 ,-1 , 0
  4479.6     .05       0    5069     .03       0    5112     .05       0
Bank Sta=5069,5112
XS Rating Curve= 0 ,0
Exp/Cntr=0.3,0.1

Type RM Length L Ch R = 1 ,11500   ,500,500,500
BEGIN DESCRIPTION:
MARSCHALL BRANCH 23.0
END DESCRIPTION:
XS GIS Cut Line= 3
       2729623.6     10174772.43      2730481.48     10174576.82
      2730881.48     10174330.23
#Sta/Elev= 30
  4120.1 1387.55  4272.7 1381.47  4320.9 1381.37  4378.7 1376.18  4406.9 1377.92
    4455 1375.99  4522.3 1376.64  4778.7  1372.2  4857.4 1373.73    4912 1363.44
  4953.7 1360.44    5035 1360.47  5050.1 1358.33  5051.1 1357.83  5093.2 1358.33
  5098.9 1360.46  5122.4 1359.84  5129.6 1361.05    5145 1366.97  5166.3 1371.71
  5224.2 1374.79  5275.1 1379.94  5340.1 1390.44    5346 1389.11  5398.1 1391.67
  5413.5 1390.45  5419.4 1391.83  5434.8 1389.68  5440.7 1390.62  5469.9 1388.93
#Mann= 3 ,-1 , 0
  4120.1     .05       0  5050.1     .03       0  5093.2     .05       0
Bank Sta=5050.1,5093.2
XS Rating Curve= 0 ,0
Exp/Cntr=0.3,0.1

Type RM Length L Ch R = 1 ,11000   ,500,500,500
BEGIN DESCRIPTION:
MARSCHALL BRANCH 22.0
END DESCRIPTION:
XS GIS Cut Line= 3
      2729605.65     10175253.12      2730629.84     10175046.62
      2731005.71     10174703.09
#Sta/Elev= 30
  3955.2 1403.68  3985.8 1399.94  4006.2  1400.7  4016.4 1397.69  4036.8 1395.77
  4087.8 1393.45  4108.3 1393.83  4331.1 1381.63  4444.9 1377.32  4534.3 1375.01
    4641 1376.84  4852.9 1369.88  4951.7 1369.01  4965.2 1368.04  4975.4 1363.89
  4982.3 1359.44  4992.1 1354.78  4993.1 1354.28  5035.2 1354.78  5070.4 1356.33
  5133.9 1355.94  5162.3 1358.86  5169.7 1360.45  5176.5 1364.02  5190.6 1366.02
  5247.4 1369.81  5360.2 1373.64  5388.6 1377.44  5431.2 1378.41  5509.2 1384.86
#Mann= 5 ,-1 , 0
  3955.2     .05       0  4951.7     .12       0  4982.3     .05       0
  4992.1     .05       0  5035.2     .05       0
Bank Sta=4992.1,5035.2
XS Rating Curve= 0 ,0
Exp/Cntr=0.3,0.1

Type RM Length L Ch R = 1 ,10500   ,500,500,500
BEGIN DESCRIPTION:
MARSCHALL BRANCH 21.0
END DESCRIPTION:
XS GIS Cut Line= 3
      2729880.68     10175678.11      2730674.19     10175516.99
      2731330.66     10175378.12
#Sta/Elev= 30
  4190.3 1392.83  4205.6 1393.48  4377.3  1389.1  4450.5 1381.92    4624 1374.64
  4685.2  1370.5  4787.2 1367.91  4817.2 1368.66    4889 1369.16  4944.8 1367.31
  4950.5 1364.03  4959.2 1356.87  4973.8 1351.36  4974.8 1350.86  5016.9 1351.36
  5052.6 1354.49  5083.3 1355.42  5139.5 1361.17  5154.8 1361.61  5165.1 1363.57
  5233.8 1367.91    5383  1373.6  5427.6 1376.41  5432.7 1375.75  5461.5  1376.7
    5527 1379.93  5543.3 1382.06  5563.7 1382.04  5604.6 1384.86    5671 1384.55
#Mann= 6 ,-1 , 0
  4190.3     .12       0  4377.3     .05       0  4817.2     .12       0
  4959.2     .05       0  4973.8     .05       0  5016.9     .05       0
Bank Sta=4973.8,5016.9
XS Rating Curve= 0 ,0
Exp/Cntr=0.3,0.1

Type RM Length L Ch R = 1 ,10000   ,500,500,500
BEGIN DESCRIPTION:
MARSCHALL BRANCH 20.0
END DESCRIPTION:
XS GIS Cut Line= 3
      2730080.71     10175828.12       2730660.5     10176015.77
      2731180.65     10175628.14
#Sta/Elev= 30
  4390.6 1384.78  4469.4 1384.22  4479.9    1381  4486.6 1380.56  4700.6 1370.93
  4817.1 1367.15  4875.9 1368.11  4889.8 1367.39  4913.1 1364.61  4939.9 1358.92
  4945.1 1359.11  4952.9 1356.98  4955.6 1350.92  4956.6 1350.42  4998.7 1350.92
    5069 1352.03  5077.4 1354.87  5083.6 1355.71    5092 1359.86  5127.5 1362.49
  5148.3 1362.71  5162.9 1364.31  5169.1 1363.54  5228.1 1365.32  5298.4 1367.45
    5313 1368.78  5355.4 1369.46  5448.6 1373.03  5563.3    1379  5648.7 1379.98
#Mann= 5 ,-1 , 0
  4390.6     .05       0  4955.6     .05       0  4998.7     .05       0
  5228.1     .12       0  5355.4     .05       0
Bank Sta=4955.6,4998.7
XS Rating Curve= 0 ,0
Exp/Cntr=0.3,0.1

Type RM Length L Ch R = 1 ,9500    ,500,500,500
BEGIN DESCRIPTION:
MARSCHALL BRANCH 19.0
END DESCRIPTION:
XS GIS Cut Line= 3
      2729939.83     10177049.98      2730876.24     10176457.14
      2731180.67     10175728.15
#Sta/Elev= 30
  3891.7 1385.29  3966.9 1387.19  4076.2 1383.74  4364.4 1369.27  4525.4 1364.08
  4610.1 1357.13  4865.3 1353.41  4871.2 1355.97  4880.5 1355.24  4886.5 1361.99
  4901.7 1354.43  4907.6 1362.45  4922.9 1354.79  4928.8 1359.53  4938.2 1356.39
  4944.1 1358.27  4959.4 1354.11  4974.6 1353.15  4977.5 1350.49  4978.5 1349.99
  5020.7 1350.49  5080.2 1351.43  5087.5 1352.34  5101.9 1358.98  5111.3 1361.34
    5230 1367.33  5376.5 1367.17    5485 1371.71  5589.6 1376.37    5790 1379.77
#Mann= 5 ,-1 , 0
  3891.7     .05       0  4977.5     .05       0  5020.7     .05       0
    5230     .12       0    5485     .05       0
Bank Sta=4977.5,5020.7
XS Rating Curve= 0 ,0
Exp/Cntr=0.3,0.1

Type RM Length L Ch R = 1 ,9000    ,500,500,500
BEGIN DESCRIPTION:
MARSCHALL BRANCH 18.0
END DESCRIPTION:
XS GIS Cut Line= 3
      2730969.16     10177055.38      2731252.44     10176782.55
      2732127.35     10175513.51
#Sta/Elev= 30
  4606.7 1375.86  4683.7 1375.43  4895.7 1363.67  4973.7 1353.71  4975.3 1348.92
  4976.3 1348.42  5022.3 1348.92    5037 1350.27  5153.3 1350.61  5159.4 1351.18
  5168.2 1355.66  5174.3 1361.05  5181.5 1362.63  5292.3 1364.71  5347.4 1368.11
  5368.3 1370.86  5448.7  1371.9  5522.6 1369.13  5623.8 1366.53  5642.1 1365.74
  5735.3 1366.39  5771.3  1366.7  5792.3 1364.63  5851.2 1368.36  5976.2 1375.45
  6013.5 1376.37  6195.3 1381.88  6281.9 1386.82  6404.3 1387.93  6541.4  1384.7
#Mann= 11 ,-1 , 0
  4606.7     .05       0  4975.3     .05       0  5022.3     .05       0
  5292.3     .12       0  5522.6     .05       0  5623.8     .12       0
  5642.1     .05       0  5735.3     .12       0  5851.2     .05       0
  5976.2     .12       0  6013.5     .05       0
Bank Sta=4975.3,5022.3
XS Rating Curve= 0 ,0
Exp/Cntr=0.3,0.1

Type RM Length L Ch R = 1 ,8500    ,500,500,500
BEGIN DESCRIPTION:
MARSCHALL BRANCH 17.0
END DESCRIPTION:
XS GIS Cut Line= 3
      2731055.65     10177153.11      2731533.83     10177184.38
      2732430.72      10176978.1
#Sta/Elev= 30
  4520.8  1378.3  4570.9 1378.19    4621 1367.85  4661.1 1365.21  4741.3 1362.71
  4851.5 1362.78  4871.6 1359.31  4891.6 1349.37  4900.3 1347.61  4905.3 1349.61
  4911.7  1347.4  4917.9 1347.12  4918.9 1346.62  4965.6 1347.12  4971.8 1348.81
  5003.5 1347.52  5027.8 1349.92    5084 1348.79  5135.3 1354.28  5155.8 1354.52
  5161.4 1356.98  5166.5 1355.62  5227.6 1364.41  5282.9 1367.39    5343 1371.23
  5428.6 1376.79  5605.1 1379.65  5761.2 1378.96  5894.6  1370.5  5920.3 1370.38
#Mann= 5 ,-1 , 0
  4520.8     .05       0  4917.9     .05       0  4965.6     .05       0
  5282.9     .12       0    5343     .05       0
Bank Sta=4917.9,4965.6
XS Rating Curve= 0 ,0
Exp/Cntr=0.3,0.1

Type RM Length L Ch R = 1 ,8000    ,500,500,500
BEGIN DESCRIPTION:
MARSCHALL BRANCH 16.0
END DESCRIPTION:
XS GIS Cut Line= 3
      2730743.42     10177602.28      2731479.56     10177668.36
       2732149.7      10177593.6
#Sta/Elev= 30
  4260.9 1376.61  4283.3  1376.7  4373.6  1371.8  4504.1 1366.36  4554.6 1366.34
  4584.5 1365.14  4594.5  1365.3  4604.5 1367.33  4614.6  1367.4  4644.7 1365.89
  4660.7 1362.07  4665.7 1362.94  4674.8 1361.52  4704.9 1360.64  4795.3 1359.23
  4845.5 1361.67  4878.1 1361.54  4925.8 1361.67    4966  1346.9  4974.8 1346.06
  4975.8 1345.56  5022.5 1346.06  5026.3 1346.88  5066.5 1346.19  5097.1 1346.87
    5147  1350.4  5182.4 1355.17  5277.8 1360.26  5475.8 1371.75  5674.3  1378.4
#Mann= 6 ,-1 , 0
  4260.9     .05       0  4878.1     .12       0  4974.8     .03       0
  5022.5     .12       0  5277.8     .12       0  5475.8     .05       0
Bank Sta=4974.8,5022.5
XS Rating Curve= 0 ,0
Exp/Cntr=0.3,0.1

Type RM Length L Ch R = 1 ,7500    ,500,500,500
BEGIN DESCRIPTION:
MARSCHALL BRANCH 15.0
END DESCRIPTION:
XS GIS Cut Line= 3
      2730955.73     10177953.13      2731449.81     10178164.76
       2731855.7     10178253.12
#Sta/Elev= 30
  4462.5 1367.45  4465.2 1367.45  4471.5 1365.08  4500.5 1362.31    4593 1358.67
  4605.7 1359.14  4636.5 1358.27  4773.1 1358.17  4821.5  1357.7    4865 1359.48
  4886.8 1359.54  4897.6 1356.98    4905 1353.88  4919.4 1351.47  4928.3 1347.85
  4941.1 1344.95  4981.2  1344.7  4982.2 1344.03  4983.2 1343.53  5028.9 1343.53
  5029.9 1344.03  5036.7 1345.57  5057.2 1345.11  5087.9 1350.32  5098.1 1351.39
  5210.7 1357.37  5253.8  1357.7    5313 1359.65  5374.4 1362.88  5415.4 1366.49
#Mann= 5 ,-1 , 0
  4462.5     .05       0  4773.1     .12       0  4928.3     .05       0
  4982.2     .03       0  5029.9     .05       0
Bank Sta=4982.2,5029.9
XS Rating Curve= 0 ,0
Exp/Cntr=0.3,0.1

Type RM Length L Ch R = 1 ,7000    ,500,500,500
BEGIN DESCRIPTION:
MARSCHALL BRANCH 14.0
END DESCRIPTION:
XS GIS Cut Line= 3
       2730905.7     10178603.11        2731398.     10178657.57
       2731905.7      10178403.1
#Sta/Elev= 30
  4504.7 1367.68  4555.1 1366.31  4695.8 1358.78    4716 1358.69  4736.6 1359.97
  4822.3 1355.47  4876.9 1357.27  4907.1 1355.92  4913.1 1354.75  4918.1 1355.84
  4927.2  1351.2  4937.3 1347.85  4957.4 1349.64  4967.5 1349.15  4972.5 1343.91
  4973.5 1343.41  5020.2 1343.91  5045.6 1345.18  5084.7 1344.08    5107 1344.68
  5120.5 1344.17  5142.8 1350.97  5179.7 1353.15  5224.3 1358.04  5308.1 1355.79
  5352.8 1356.54  5425.4 1359.37  5509.2 1365.83  5537.2 1366.45  5567.9 1368.33
#Mann= 3 ,-1 , 0
  4504.7     .05       0  4972.5     .03       0  5020.2     .05       0
Bank Sta=4972.5,5020.2
XS Rating Curve= 0 ,0
Exp/Cntr=0.3,0.1

Type RM Length L Ch R = 1 ,6500    ,500,500,500
BEGIN DESCRIPTION:
MARSCHALL BRANCH 13.0
END DESCRIPTION:
XS GIS Cut Line= 3
      2730755.64     10179303.12      2731613.31     10179102.61
       2732005.7     10178603.09
#Sta/Elev= 30
  4119.2 1374.61  4150.1 1371.97    4237 1368.03  4252.8 1365.91  4270.6 1364.73
  4354.1 1361.46  4478.7 1358.36  4550.6 1359.83  4606.3 1359.12  4704.6 1357.34
    4711 1356.41  4739.7 1356.55  4838.1 1357.32  4899.7 1356.41  4933.8 1353.86
  4961.4 1350.54  4971.2 1348.12  4974.8 1342.98  4975.8 1342.48  5022.6 1342.98
  5023.3 1344.61  5029.6 1344.82  5064.9 1343.37  5095.4 1343.31  5143.5 1344.44
  5178.8 1352.44  5222.1  1354.6  5315.2 1354.79  5493.3 1362.05  5635.2 1364.76
#Mann= 8 ,-1 , 0
  4119.2     .12       0    4237     .05       0  4354.1     .12       0
  4606.3     .05       0  4739.7     .12       0  4974.8     .07       0
  5022.6     .12       0  5095.4     .05       0
Bank Sta=4974.8,5022.6
XS Rating Curve= 0 ,0
Exp/Cntr=0.3,0.1

Type RM Length L Ch R = 1 ,6000    ,500,500,500
BEGIN DESCRIPTION:
MARSCHALL BRANCH 12.0
END DESCRIPTION:
XS GIS Cut Line= 3
      2731605.67     10179703.12      2731974.46     10179430.69
      2732155.69      10178603.1
#Sta/Elev= 30
  4541.5 1362.87  4634.4 1360.02  4705.4 1355.55  4755.5 1353.85  4845.7 1353.58
  4864.1 1353.44  4914.2 1348.25  4935.1 1347.88  4949.7 1346.57  4955.9 1344.21
  4964.2 1343.05  4996.7 1342.56    5018 1342.18  5026.1 1343.94  5058.9 1344.31
  5099.9 1343.68    5100 1342.11    5101 1341.61  5148.1 1342.11  5161.3 1344.51
    5173 1344.98    5192 1348.82  5211.7 1351.41  5388.7 1355.92  5491.7 1357.86
  5561.5  1359.2  5594.8 1359.99  5694.5 1362.81  5775.3 1364.36  5847.2 1365.65
#Mann= 11 ,-1 , 0
  4541.5     .05       0  4845.7     .12       0  4996.7     .05       0
    5100     .05       0  5148.1     .05       0  5388.7     .12       0
  5491.7     .05       0  5561.5     .12       0  5594.8     .05       0
  5694.5     .12       0  5775.3     .05       0
Bank Sta=5100,5148.1
XS Rating Curve= 0 ,0
Exp/Cntr=0.3,0.1

Type RM Length L Ch R = 1 ,5500    ,500,500,500
BEGIN DESCRIPTION:
MARSCHALL BRANCH 11.0
END DESCRIPTION:
XS GIS Cut Line= 3
      2731905.65     10179953.13      2732392.12     10179685.78
      2733055.67     10179003.13
#Sta/Elev= 30
  4444.9 1364.01  4664.8 1351.48  4762.8 1351.59  4828.1 1344.04  4882.5 1344.98
  4958.9 1340.78  5011.5 1340.67  5029.8 1340.01  5030.8 1339.51    5078 1340.01
  5082.2 1347.04  5108.8 1350.06  5181.2 1353.41  5267.8 1352.07  5375.9 1352.02
  5529.6 1349.95    5563 1345.88  5591.3  1350.8  5633.7  1352.8  5647.9  1350.6
  5704.5 1355.72  5718.6 1354.43  5725.8 1356.54  5732.8 1355.37  5739.9 1356.87
  5746.9 1354.97  5775.2 1359.31  5796.5 1359.21  5860.1 1366.07    5952  1368.6
#Mann= 8 ,-1 , 0
  4444.9     .05       0  4664.8     .12       0  4882.5     .05       0
  5011.5     .05       0  5108.8     .12       0  5267.8     .05       0
  5375.9     .12       0  5529.6     .05       0
Bank Sta=5029.8,5078
XS Rating Curve= 0 ,0
Exp/Cntr=0.3,0.1

Type RM Length L Ch R = 1 ,5000    ,500,500,500
BEGIN DESCRIPTION:
MARSCHALL BRANCH 10.0
END DESCRIPTION:
XS GIS Cut Line= 3
      2732023.16     10180273.93      2732781.43     10179980.69
      2733495.17     10179251.59
#Sta/Elev= 30
    4187 1358.76  4306.3 1356.04  4315.8 1354.71  4554.3 1351.31  4607.9 1348.42
  4629.3 1349.75  4654.3 1346.92    4706 1346.48  4785.1 1341.56  4874.3 1339.87
  4886.6 1340.91  4929.5 1339.65  4972.4 1339.75  4984.3 1338.34  4985.3 1337.84
  5032.5 1338.34  5057.9 1339.66  5100.3 1338.92  5121.6 1342.87    5171    1347
  5230.1 1346.05  5312.5 1347.65  5377.8 1344.27  5397.3 1343.06  5432.6 1344.97
  5446.8 1342.25  5538.8 1345.01  5581.2 1348.84  5800.4 1352.03  6020.3 1358.94
#Mann= 8 ,-1 , 0
    4187     .05       0  4306.3     .12       0  4315.8     .05       0
  4654.3     .12       0  4874.3     .05       0  4929.5     .05       0
  5230.1     .12       0  5377.8     .05       0
Bank Sta=4984.3,5032.5
XS Rating Curve= 0 ,0
Exp/Cntr=0.3,0.1

Type RM Length L Ch R = 1 ,4500    ,500,500,500
BEGIN DESCRIPTION:
MARSCHALL BRANCH 9.0
END DESCRIPTION:
XS GIS Cut Line= 3
      2732465.87     10181190.62      2733195.41     10180227.66
      2733651.06     10179642.68
#Sta/Elev= 30
  3791.9 1355.51  3832.8 1357.57  3882.8 1353.81  4042.6 1350.13  4228.5 1349.22
  4481.9 1344.01  4540.2 1336.03  4586.7 1336.02  4596.4 1336.43  4610.9 1341.47
  4660.8 1346.27  4725.3 1345.29  4767.3 1340.94  4944.8  1335.3  4989.5 1335.48
  5000.7 1333.91  5001.7 1333.41  5048.9 1333.91  5053.8 1335.98  5081.8 1336.37
  5095.4 1339.67  5185.3 1343.75    5232 1343.29  5259.3    1340  5305.8 1340.48
  5373.4 1344.78  5416.6 1352.79  5466.3 1356.88  5580.3 1361.26  5741.5 1362.63
#Mann= 9 ,-1 , 0
  3791.9     .05       0  4042.6     .12       0  4228.5     .05       0
  4586.7     .12       0  4944.8     .05       0  5000.7     .05       0
  5048.9     .05       0  5185.3     .12       0  5305.8     .05       0
Bank Sta=5000.7,5048.9
XS Rating Curve= 0 ,0
Exp/Cntr=0.3,0.1

Type RM Length L Ch R = 1 ,4000    ,500,500,500
BEGIN DESCRIPTION:
MARSCHALL BRANCH 8.0
END DESCRIPTION:
XS GIS Cut Line= 3
      2733116.93     10182003.11      2733551.06     10180542.56
      2733764.26     10180041.54
#Sta/Elev= 30
  3476.3 1358.13  3695.1 1359.42  3883.2 1351.19  3976.3 1349.41  4086.4 1351.18
  4152.8 1343.84    4158 1344.73  4196.4 1338.15  4224.4 1338.94  4249.3 1335.89
  4257.6 1335.36  4269.2 1339.07  4279.6 1339.67  4415.2 1339.72    4553 1345.18
  4634.3 1345.82  4728.2 1342.36  4811.6  1341.9  4853.2 1337.55  4874.2 1329.74
  4975.1 1329.28  4976.1 1328.78  5023.5 1329.28  5078.3 1330.88  5172.8 1330.79
  5201.9 1336.47  5325.4 1352.02    5331 1354.67  5401.5 1361.59  5544.5 1361.02
#Mann= 4 ,-1 , 0
  3476.3     .05       0  4249.3     .12       0    4553     .05       0
  5078.3     .05       0
Bank Sta=4975.1,5023.5
XS Rating Curve= 0 ,0
Exp/Cntr=0.3,0.1

Type RM Length L Ch R = 1 ,3500    ,500,500,500
BEGIN DESCRIPTION:
MARSCHALL BRANCH 7.0
END DESCRIPTION:
XS GIS Cut Line= 3
      2733564.61     10181630.07      2733937.05     10180828.35
      2734154.84     10180197.91
#Sta/Elev= 30
    4116 1350.12  4341.4 1343.12  4364.3 1339.78  4369.8  1340.8  4377.3 1336.82
  4387.1 1334.22  4392.7 1335.62    4410 1331.43  4421.4 1331.15  4438.4 1334.43
  4454.5 1334.79  4619.9 1334.45    4770 1336.58  4838.7 1332.63  4873.5 1324.88
  4895.5 1326.12  4976.6 1324.59  4977.9 1323.69  5034.5 1324.59  5036.9 1327.61
  5130.4 1335.93  5206.6 1347.54  5255.1 1350.17  5301.8  1347.6  5343.4 1350.23
  5386.4 1359.27  5481.6 1369.88  5587.4 1374.32  5655.2 1373.46    5667 1372.04
#Mann= 3 ,-1 , 0
    4116     .05       0  4976.6     .07       0  5034.5     .05       0
Bank Sta=4976.6,5034.5
XS Rating Curve= 0 ,0
Exp/Cntr=0.3,0.1

Type RM Length L Ch R = 1 ,3000    ,500,500,500
BEGIN DESCRIPTION:
MARSCHALL BRANCH 6.0
END DESCRIPTION:
XS GIS Cut Line= 3
      2734505.69     10181703.13      2734296.03     10181065.41
      2734255.68      10180553.1
#Sta/Elev= 30
  4328.7    1345  4360.3  1340.7  4408.2 1341.39  4528.7 1336.34  4560.3 1333.85
  4604.3 1333.47  4667.9 1327.08  4686.6 1326.36  4699.7 1328.19  4726.2 1328.45
    4758 1326.71  4763.3 1327.82  4781.4 1323.03  4783.7  1320.7  4785.1  1319.8
  4840.7  1319.8  4842.2  1320.7  4844.5 1323.45  5042.4 1324.61  5067.8 1328.76
  5072.8 1328.19  5092.6 1331.01  5152.8 1332.45  5196.7 1335.85    5223 1340.04
  5293.2 1342.25  5363.4 1341.25  5483.8 1347.81  5493.8 1348.59  5513.9 1352.95
#Mann= 3 ,-1 , 0
  4328.7     .05       0  4783.7     .07       0  4842.2     .05       0
Bank Sta=4783.7,4842.2
XS Rating Curve= 0 ,0
Exp/Cntr=0.3,0.1

Type RM Length L Ch R = 1 ,2500    ,500,500,500
BEGIN DESCRIPTION:
MARSCHALL BRANCH 5.0
END DESCRIPTION:
XS GIS Cut Line= 3
      2734555.68     10181653.12      2734754.92      10181239.4
      2735005.69      10180903.1
#Sta/Elev= 30
  4540.8 1340.99  4577.5 1339.12  4617.2 1335.33  4645.4 1335.88  4651.8 1334.31
    4668    1333  4809.3 1329.84  4826.4 1327.85  4854.5 1326.73  4894.2 1328.55
  4899.8 1328.21  4916.9 1320.14  4951.5 1319.26  4955.4 1318.45  4956.8 1317.55
  5012.6 1317.55    5014 1318.45  5020.2 1319.44  5082.7 1319.11  5091.1 1320.26
  5132.8 1319.68  5155.7 1323.88    5162 1323.39  5176.6 1327.38  5241.2 1335.94
  5262.1 1337.47  5276.7 1339.94  5347.5 1344.93    5383 1350.15  5419.5 1353.16
#Mann= 3 ,-1 , 0
  4540.8     .05       0  4955.4     .07       0    5014     .05       0
Bank Sta=4955.4,5014
XS Rating Curve= 0 ,0
Exp/Cntr=0.3,0.1

Type RM Length L Ch R = 1 ,2000    ,500,500,500
BEGIN DESCRIPTION:
MARSCHALL BRANCH 4.0
END DESCRIPTION:
XS GIS Cut Line= 3
      2735305.68     10182203.07      2735238.33     10181248.34
      2735205.69     10181053.15
#Sta/Elev= 30
  4042.9 1375.11    4093 1372.67  4133.1  1366.6  4213.3  1359.3  4233.3 1353.68
  4252.2 1353.19  4263.4 1349.84  4283.5 1350.18  4313.5 1347.79  4398.4 1336.67
  4413.8 1332.81  4453.9 1328.12    4484 1328.07  4574.2 1332.53  4614.3 1331.52
  4664.4 1327.72  4744.6  1327.5  4784.7 1325.43  4834.8 1322.26  4884.9 1321.17
    4915 1316.76  4975.2  1317.5  5019.3 1315.68  5020.7 1314.78  5077.9 1315.68
  5086.4 1324.26  5104.3 1332.17  5116.8 1334.79    5165 1335.76  5197.9 1340.59
#Mann= 4 ,-1 , 0
  4042.9     .07       0  4784.7     .07       0  5019.3    .055       0
  5077.9    .055       0
Bank Sta=5019.3,5077.9
XS Rating Curve= 0 ,0
Exp/Cntr=0.3,0.1

Type RM Length L Ch R = 1 ,1500    ,500,500,500
BEGIN DESCRIPTION:
MARSCHALL BRANCH 3.0
END DESCRIPTION:
XS GIS Cut Line= 3
      2735455.68     10182353.12       2735706.5       10181404.
      2735805.67     10181053.15
#Sta/Elev= 30
  4018.3 1384.18  4101.1 1371.67  4111.2 1359.73  4121.7 1353.79  4132.1 1353.01
  4151.4 1357.89  4156.6 1352.07  4163.1 1352.07  4191.7 1361.17  4196.9 1350.61
  4204.5 1355.76  4225.2 1358.77  4256.2 1348.41  4266.5  1351.4  4277.4  1346.7
  4307.3 1344.32  4312.5  1341.7  4318.3 1343.74  4566.5 1331.28  4866.5 1323.04
  4907.8 1314.34  4940.5 1313.54  4941.9 1312.64  4999.2 1313.54  5021.7 1314.47
  5049.9 1320.57  5089.1 1320.56  5123.1 1325.59  5208.8 1331.88  5364.6 1349.22
#Mann= 3 ,-1 , 0
  4018.3     .07       0  4940.5     .07       0  4999.2     .07       0
Bank Sta=4940.5,4999.2
XS Rating Curve= 0 ,0
Exp/Cntr=0.3,0.1

Type RM Length L Ch R = 1 ,1000    ,193,193,193
BEGIN DESCRIPTION:
MARSCHALL BRANCH 2.0
END DESCRIPTION:
XS GIS Cut Line= 3
      2735596.67     10182381.11       2736184.1     10181514.67
      2735921.01     10180990.04
#Sta/Elev= 30
  3953.2 1363.81  4030.5 1356.39  4087.4 1346.49  4102.4 1350.76  4123.3 1344.91
  4138.3 1347.71  4153.2 1346.05  4159.3  1342.2  4168.2 1344.25  4174.2 1340.63
  4189.2 1342.55  4195.2 1338.26  4204.1 1338.99  4210.2 1335.06  4246.1 1329.46
  4368.9 1327.82  4425.8 1323.56  4692.4  1321.2  4699.8 1325.97  4785.3 1326.73
    4908 1318.87  4929.4  1312.5  4983.7 1310.75  4985.1 1309.85  5042.4 1310.75
  5057.8 1312.89  5096.8  1320.1  5169.5 1325.59  5253.2 1326.69  5586.9 1353.39
#Mann= 3 ,-1 , 0
  3953.2     .07       0  4983.7     .07       0  5057.8     .07       0
Bank Sta=4983.7,5042.4
XS Rating Curve= 0 ,0
Exp/Cntr=0.3,0.1

Type RM Length L Ch R = 1 ,807     ,229,229,229
BEGIN DESCRIPTION:
Mapping XS 7a142d09
END DESCRIPTION:
XS GIS Cut Line= 6
      2735494.62      10182648.8      2735821.02     10182551.57
      2736376.58      10181759.9      2736362.69     10181419.63
      2736064.08      10180947.4      2735898.25     10180636.47
#Sta/Elev= 30
  3493.2 1370.17  3530.7 1366.43  3546.5 1360.32  3563.9 1348.39  3602.3 1348.72
  3635.4 1343.86  3661.3 1344.73  3673.8 1349.71    3707 1348.71  3734.3 1339.74
  3773.3 1336.24  3929.6 1336.19  3951.5 1338.93  3972.4 1320.27  4109.3 1323.93
  4827.7 1327.08  4857.8 1327.36  4877.8 1320.68  4917.8 1312.87  5007.9 1310.62
    5088 1320.02  5144.3 1325.28  5447.8 1323.81  5535.9 1327.87  5599.5  1336.2
  5709.1  1343.5  5813.2 1337.53  5841.1 1345.56    5923 1358.19  6052.6 1369.78
#Mann= 4 ,-1 , 0
  3493.2     .05       0  4137.3     .03       0  4827.7    .045       0
  5535.9     .05       0
Bank Sta=4877.8,5088
XS Rating Curve= 0 ,0
Exp/Cntr=0.3,0.1

Type RM Length L Ch R = 1 ,578     ,198,198,198
BEGIN DESCRIPTION:
Mapping XS 4c84ac10
END DESCRIPTION:
XS GIS Cut Line= 5
      2735705.61     10182983.56       2736161.3     10182294.63
      2736591.86     10181614.07      2736584.91      10181259.9
      2735974.95     10180476.65
#Sta/Elev= 30
  3374.1 1346.66  3662.4    1337  3749.1 1340.33  3872.5 1338.78    4032 1330.36
  4189.9 1328.79  4343.3 1332.88  4805.4  1333.4  4877.3 1337.43  4892.6 1332.97
  4907.8 1319.77  4913.8 1319.71  4923.1 1315.15  4971.4 1310.06  5026.4  1311.1
  5096.4 1319.52  5166.4 1324.49  5246.4 1319.68  5316.4 1328.49    5414 1331.47
  5470.1 1326.54  5606.7 1335.31  5855.5 1328.22  6019.3 1338.43  6048.2 1343.45
  6162.2 1345.95  6176.7 1348.06  6197.5 1357.92  6218.3  1360.9  6352.4 1372.42
#Mann= 4 ,-1 , 0
  3374.1    .045       0  4907.8     .03       0  5166.4    .045       0
  5316.4     .05       0
Bank Sta=4913.8,5096.4
XS Rating Curve= 0 ,0
Exp/Cntr=0.3,0.1

Type RM Length L Ch R = 1 ,380     ,234,234,234
BEGIN DESCRIPTION:
Mapping XS 9dc69405
END DESCRIPTION:
XS GIS Cut Line= 6
      2735790.66     10182962.26      2736182.14     10182468.24
      2736765.47     10181718.24      2736834.91     10181426.57
      2736730.75      10181009.9      2736105.76     10180482.13
#Sta/Elev= 30
  3332.8 1345.14    3414  1348.6  3556.6 1337.04  3641.5 1341.77  3883.5 1337.52
  4096.9 1326.71  4418.1  1332.4    4590 1326.11  4666.9 1343.99  4739.3 1341.19
  4859.7 1348.78  4881.8 1343.55  4888.6 1336.58    4895 1340.74  4913.3 1334.83
  4918.5    1325  4934.9 1312.12  4994.9 1309.96  4996.4 1309.06  5053.7 1309.96
  5061.3  1315.9  5124.1 1321.19  5319.7 1317.47  5473.6 1324.92    5722 1331.96
  5898.9 1326.13  6105.6 1338.78  6290.2 1333.61  6409.9 1338.16  6460.6 1346.32
#Mann= 3 ,-1 , 0
  3332.8     .05       0  4994.9     .03       0  5473.6     .05       0
Bank Sta=4994.9,5053.7
XS Rating Curve= 0 ,0
Exp/Cntr=0.3,0.1

Type RM Length L Ch R = 1 ,146     ,0,0,0
BEGIN DESCRIPTION:
MARSCHALL BRANCH 1.0
END DESCRIPTION:
XS GIS Cut Line= 3
      2736140.44     10182822.44      2737005.25       10181705.
      2737890.46     10181134.91
#Sta/Elev= 30
    3587 1342.86  3683.2 1337.69  3832.6 1335.58  3940.2 1327.47  4117.2 1324.57
  4145.9 1330.08  4210.2 1323.64  4303.4 1330.54  4423.9 1330.03  4481.8 1338.58
  4496.3 1346.45  4517.1 1365.81  4537.9 1372.93    4710    1360  4787.4 1362.55
  4809.6 1348.71  4844.9 1315.84  4865.7 1309.81  4938.2 1311.83    4958 1307.39
  4959.5 1306.39    5018 1307.39  5333.6 1312.98    5545  1324.6  5644.7  1330.1
  5696.2 1328.51  5711.4 1324.26  5726.8 1327.85  5753.6  1332.5  6052.9 1336.59
#Mann= 4 ,-1 , 0
    3587     .05       0    4958     .03       0    5545     .05       0
  5726.8     .05       0
#XS Ineff= 2 , 0
         4538.25 1373.44 5827.87         1334.59
Permanent Ineff=
       F       F
Bank Sta=4958,5018
XS Rating Curve= 0 ,0
Exp/Cntr=0.3,0.1
Stream Node=MARSCHALL BRANCH,Reach-1         , 0 , 0 ,Upstream end
Stream Node=MARSCHALL BRANCH,Reach-1         , 0 , 1 ,Downstream end

Chan Stop Cuts=-1
Use User Specified Reach Order=0
Composite Channel Slope=5
