--- LITTLE LLANO 052.prj (project) ---

Proj Title=LITTLE LLANO 052 Base Level Engineering
Current Plan=p01
Default Exp/Contr=0.3,0.1
English Units
Geom File=g01
Flow File=f01
Plan File=p01
BEGIN DESCRIPTION:
LITTLE LLANO 052
END DESCRIPTION:

--- LITTLE LLANO 052.p01 (plan) ---

Plan Title=Multiple Run
Short Identifier=Multiple
Geom File=g01
Flow File=f01
Subcritical Flow
K Sum by GR= 0
Std Step Tol= 0.01
Critical Tol= 0.01
Num of Std Step Trials= 20
Max Error Tol= 0.3
Flow Tol Ratio= 0.001
Split Flow NTrial= 30
Split Flow Tol= 0.02
Split Flow Ratio= 0.02
Log Output Level= 0
Friction Slope Method= 1
Unsteady Friction Slope Method= 2
Unsteady Bridges Friction Slope Method= 1
Parabolic Critical Depth
Global Vel Dist=  1 , 1 , 1
Global Log Level= 0
CheckData=True
Encroach Param= -1, 0, 0, 0
BEGIN DESCRIPTION:
Multiple Run
END DESCRIPTION:

--- LITTLE LLANO 052.f01 (steady flow) ---

Flow Title=Multiple
Number of Profiles=7
Profile Names=10-year,25-year,50-year,1pct_min,100-year,1pct_plu,500-year
River Rch & RM= LITTLE LLANO 052,Reach-1,27001
     410     658    1175     949    1615    2749    2294
River Rch & RM= LITTLE LLANO 052,Reach-1,19230
     721    1206    1991    1474    2762    5177    3875
River Rch & RM= LITTLE LLANO 052,Reach-1,12839
    1102    1907    2886    1983    4025    8170    5600
River Rch & RM= LITTLE LLANO 052,Reach-1,3823
    1271    2223    3290    2216    4600    9551    6384
Boundary for River Rch & Prof#=LITTLE LLANO 052,Reach-1,1
Up Type=0
Dn Type=3
Dn Slope=0.005
Boundary for River Rch & Prof#=LITTLE LLANO 052,Reach-1,2
Up Type=0
Dn Type=3
Dn Slope=0.005
Boundary for River Rch & Prof#=LITTLE LLANO 052,Reach-1,3
Up Type=0
Dn Type=3
Dn Slope=0.005
Boundary for River Rch & Prof#=LITTLE LLANO 052,Reach-1,4
Up Type=0
Dn Type=3
Dn Slope=0.005
Boundary for River Rch & Prof#=LITTLE LLANO 052,Reach-1,5
Up Type=0
Dn Type=3
Dn Slope=0.005
Boundary for River Rch & Prof#=LITTLE LLANO 052,Reach-1,6
Up Type=0
Dn Type=3
Dn Slope=0.005
Boundary for River Rch & Prof#=LITTLE LLANO 052,Reach-1,7
Up Type=0
Dn Type=3
Dn Slope=0.005

--- LITTLE LLANO 052.g01 (geometry) ---

Geom Title=Existing Conditions

River Reach=LITTLE LLANO 052,Reach-1
Reach XY= 30
      2828584.50     10269412.00      2829148.25     10267916.00
      2828851.00     10267342.00      2829163.50     10265897.00
      2829134.00     10264698.00      2830009.00     10264711.00
      2830052.00     10264487.00      2830552.00     10264582.00
      2830958.25     10264314.00      2831300.50     10264619.00
      2832178.25     10264232.00      2832488.00     10264433.00
      2833859.25     10263877.00      2834596.25     10264056.00
      2834387.75     10264370.00      2835437.25     10264407.00
      2835981.50     10263926.00      2837656.00     10263956.00
      2838580.50     10263366.00      2839824.00     10264478.00
      2839611.75     10263757.00      2840350.00     10263411.00
      2841005.00     10263580.00      2842578.00     10263420.00
      2842774.50     10262957.00      2842338.25     10262917.00
      2842347.50     10262684.00      2842818.75     10262125.00
      2843143.00     10262454.00      2844230.00     10262580.00

Type RM Length L Ch R = 1,27001,471,471,471
BEGIN DESCRIPTION:
LITTLE LLANO 052 54.0
END DESCRIPTION:
XS GIS Cut Line= 3
      2828805.64     10269203.10      2828635.75     10269149.00
      2828405.73     10269203.10
#Sta/Elev= 30
  4821.7 1233.46  4832.2 1231.96  4843.0 1228.87  4853.1 1227.47  4875.2 1222.92
  4939.7 1212.19  4947.6 1211.15  4958.1 1211.58  4995.4 1207.69  4995.7 1207.19
  4999.2 1207.19  4999.4 1207.69  5010.3 1208.82  5020.6 1211.32  5030.9 1211.47
  5051.4 1213.17  5061.7 1215.70  5085.4 1219.53  5122.7 1222.88  5143.9 1225.51
  5154.2 1227.55  5170.2 1233.38  5175.3 1234.05  5185.0 1238.18  5205.5 1241.23
  5212.6 1244.50  5217.7 1245.53  5226.1 1249.51  5233.8 1251.41  5236.3 1251.41
#Mann=3,-1,0
  4821.7    0.05       0  4995.4    0.03       0  4999.4    0.05       0
Bank Sta=4995.4,4999.4
Exp/Cntr=0.3,0.1

Type RM Length L Ch R = 1,26530,405,405,405
BEGIN DESCRIPTION:
LITTLE LLANO 052 53.0
END DESCRIPTION:
XS GIS Cut Line= 3
      2829055.67     10268753.11      2828735.75     10268692.00
      2828455.64     10268753.12
#Sta/Elev= 30
  4674.3 1225.92  4700.3 1224.06  4745.5 1217.54  4809.6 1211.84  4837.2 1208.06
  4861.7 1205.94  4877.9 1205.90  4908.4 1202.13  4913.8 1200.78  4949.2 1197.34
  4971.0 1192.90  4979.7 1194.86  4989.9 1194.48  4997.5 1191.19  5008.3 1191.09
  5008.6 1190.59  5012.3 1191.09  5020.5 1192.72  5027.2 1195.55  5071.1 1199.83
  5102.4 1201.39  5125.2 1204.81  5133.1 1208.62  5184.3 1217.08  5255.9 1236.70
  5262.1 1239.37  5267.3 1239.84  5276.4 1242.26  5284.1 1245.98  5286.7 1245.98
#Mann=3,-1,0
  4674.3    0.05       0  5008.3    0.03       0  5012.3    0.05       0
Bank Sta=5008.3,5012.3
Exp/Cntr=0.3,0.1

Type RM Length L Ch R = 1,26125,418,418,418
BEGIN DESCRIPTION:
LITTLE LLANO 052 52.0
END DESCRIPTION:
XS GIS Cut Line= 3
      2829155.65     10268603.08      2828880.75     10268327.00
      2828605.69     10268353.11
#Sta/Elev= 30
  4610.4 1221.83  4624.5 1220.31  4645.7 1215.91  4652.8 1215.66  4659.8 1213.56
  4709.3 1207.53  4715.9 1207.53  4723.5 1205.77  4730.6 1206.31  4737.6 1204.30
  4744.7 1204.05  4765.9 1200.50  4794.2 1197.19  4864.9 1191.07  4920.6 1187.85
  4978.0 1182.51  4985.1 1182.44  4992.2 1180.72  5003.1 1180.16  5003.3 1179.66
  5007.1 1180.16  5010.9 1182.26  5025.2 1184.41  5119.1 1192.14  5125.6 1193.57
  5155.8 1196.84  5195.9 1204.83  5216.0 1206.77  5246.2 1213.25  5276.3 1217.52
#Mann=5,-1,0
  4610.4    0.05       0  4715.9    0.12       0  4920.6    0.05       0
  5003.1    0.03       0  5007.1    0.05       0
Bank Sta=5003.1,5007.1
Exp/Cntr=0.3,0.1

Type RM Length L Ch R = 1,25707,473,473,473
BEGIN DESCRIPTION:
LITTLE LLANO 052 51.0
END DESCRIPTION:
XS GIS Cut Line= 3
      2829155.66     10268053.09      2829064.75     10267967.00
      2828955.67     10268003.12
#Sta/Elev= 30
  4874.8 1179.43  4878.2 1179.43  4881.8 1178.66  4896.0 1178.05  4902.9 1177.22
  4910.2 1177.16  4917.0 1177.31  4924.3 1175.80  4931.2 1174.85  4938.5 1174.25
  4973.7 1170.37  4980.9 1170.26  4987.8 1168.76  4995.1 1168.52  4997.2 1167.10
  4997.4 1166.60  5000.9 1166.60  5001.2 1167.10  5003.9 1168.52  5009.5 1168.25
  5030.4 1168.19  5051.7 1171.00  5062.1 1172.14  5067.3 1171.11  5083.3 1173.10
  5093.8 1174.61  5099.0 1173.28  5104.4 1176.56  5112.3 1178.57  5114.9 1178.57
#Mann=3,-1,0
  4874.8    0.05       0  4997.2    0.05       0  5001.2    0.05       0
Bank Sta=4997.2,5001.2
Exp/Cntr=0.3,0.1

Type RM Length L Ch R = 1,25234,496,496,496
BEGIN DESCRIPTION:
LITTLE LLANO 052 50.0
END DESCRIPTION:
XS GIS Cut Line= 3
      2829205.71     10267603.12      2829062.00     10267563.00
      2828805.70     10267853.10
#Sta/Elev= 30
  4850.8 1170.10  4902.1 1166.02  4907.3 1166.51  4915.7 1165.20  4941.4 1160.93
  4946.6 1161.31  4975.4 1158.61  4980.8 1157.22  5002.4 1156.78  5002.7 1156.28
  5006.4 1156.78  5012.0 1158.30  5018.6 1157.72  5026.2 1159.06  5032.9 1157.81
  5047.1 1160.15  5053.7 1159.38  5061.3 1160.23  5068.0 1159.63  5075.5 1160.59
  5082.2 1160.05  5089.7 1160.98  5121.8 1161.44  5132.4 1161.93  5153.3 1160.64
  5174.2 1160.97  5196.0 1162.19  5202.7 1163.80  5259.5 1166.50  5387.1 1174.48
#Mann=5,-1,0
  4850.8    0.05       0  4915.7    0.12       0  5002.4    0.07       0
  5006.4    0.12       0  5121.8    0.05       0
Bank Sta=5002.4,5006.4
Exp/Cntr=0.3,0.1

Type RM Length L Ch R = 1,24738,490,490,490
BEGIN DESCRIPTION:
LITTLE LLANO 052 49.0
END DESCRIPTION:
XS GIS Cut Line= 3
      2829005.65     10267203.11      2828902.25     10267188.00
      2828605.70     10267153.11
#Sta/Elev= 30
  4895.5 1152.72  4915.7 1150.70  4925.4 1149.97  4930.4 1150.00  4935.9 1149.03
  4966.2 1147.78  4976.3 1146.54  4986.4 1142.79  4995.4 1141.68  4997.6 1141.04
  4997.9 1140.54  5001.4 1140.54  5001.6 1141.04  5016.7 1144.19  5067.0 1148.65
  5083.4 1149.92  5088.4 1149.80  5137.5 1153.91  5157.6 1156.11  5171.5 1156.82
  5177.8 1157.67  5187.9 1158.23  5238.2 1163.62  5248.3 1165.22  5254.6 1167.42
  5259.6 1166.73  5278.5 1171.38  5288.5 1174.24  5296.1 1178.03  5298.6 1178.03
#Mann=3,-1,0
  4895.5    0.05       0  4997.6    0.05       0  5001.6    0.05       0
Bank Sta=4997.6,5001.6
Exp/Cntr=0.3,0.1

Type RM Length L Ch R = 1,24248,467,467,467
BEGIN DESCRIPTION:
LITTLE LLANO 052 48.0
END DESCRIPTION:
XS GIS Cut Line= 3
      2829255.69     10266703.11      2828949.00     10266724.00
      2828855.64     10266753.13
#Sta/Elev= 30
  4692.6 1158.72  4752.7 1153.56  4767.0 1151.94  4782.8 1149.47  4812.9 1146.49
  4832.9 1143.41  4843.0 1142.51  4859.3 1140.19  4863.0 1139.66  4873.0 1141.61
  4963.2 1139.12  4973.3 1138.40  4983.3 1136.82  4991.3 1133.71  4991.6 1133.21
  4995.1 1133.21  4995.3 1133.71  4999.2 1134.87  5004.4 1134.87  5011.3 1138.36
  5016.5 1138.78  5024.4 1141.71  5034.9 1143.31  5043.8 1144.38  5049.0 1144.29
  5055.8 1145.62  5076.3 1147.19  5081.5 1146.83  5087.3 1147.27  5097.8 1147.15
#Mann=4,-1,0
  4692.6    0.12       0  4859.3    0.05       0  4991.3    0.05       0
  4995.3    0.05       0
Bank Sta=4991.3,4995.3
Exp/Cntr=0.3,0.1

Type RM Length L Ch R = 1,23781,465,465,465
BEGIN DESCRIPTION:
LITTLE LLANO 052 47.0
END DESCRIPTION:
XS GIS Cut Line= 3
      2829255.66     10266403.11      2828938.50     10266368.00
      2828855.73     10266353.12
#Sta/Elev= 30
  4680.9 1156.79  4701.0 1155.74  4721.1 1152.55  4726.2 1150.76  4731.3 1152.47
  4741.2 1151.21  4751.3 1149.56  4791.6 1138.97  4801.6 1137.19  4811.7 1137.31
  4831.8 1135.92  4841.9 1134.02  4862.0 1133.64  4872.0 1134.14  4892.2 1131.29
  4907.7 1130.59  4912.7 1129.53  4920.3 1129.25  4920.6 1128.75  4924.1 1128.75
  4924.3 1129.25  4930.2 1129.68  4942.5 1130.50  4992.8 1131.19  5004.0 1130.49
  5013.0 1132.71  5023.2 1136.82  5033.3 1138.64  5057.3 1142.22  5084.1 1143.59
#Mann=4,-1,0
  4680.9    0.12       0  4920.3    0.05       0  4924.3    0.12       0
  4930.2    0.05       0
Bank Sta=4920.3,4924.3
Exp/Cntr=0.3,0.1

Type RM Length L Ch R = 1,23316,462,462,462
BEGIN DESCRIPTION:
LITTLE LLANO 052 46.0
END DESCRIPTION:
XS GIS Cut Line= 3
      2829355.65     10266253.09      2829032.25     10266053.00
      2828755.71     10266153.10
#Sta/Elev= 30
  4619.7 1169.63  4654.9 1163.24  4765.8 1147.53  4779.8 1144.17  4801.1 1144.39
  4822.3 1140.87  4837.7 1136.45  4880.2 1133.26  4889.8 1130.98  4925.4 1130.43
  4988.1 1125.97  4994.1 1125.93  5005.0 1124.95  5005.2 1124.45  5009.0 1124.95
  5013.7 1127.97  5020.6 1126.98  5069.6 1129.96  5074.9 1132.88  5100.3 1131.93
  5105.6 1134.41  5130.9 1131.56  5161.6 1135.23  5166.9 1133.08  5186.9 1135.98
  5192.2 1134.06  5217.5 1138.07  5222.8 1136.73  5248.2 1144.42  5294.1 1147.89
#Mann=7,-1,0
  4619.7    0.05       0  4765.8    0.12       0  4988.1    0.05       0
  4994.1    0.12       0  5005.0    0.07       0  5009.0    0.12       0
  5020.6    0.05       0
Bank Sta=5005,5009
Exp/Cntr=0.3,0.1

Type RM Length L Ch R = 1,22854,450,450,450
BEGIN DESCRIPTION:
LITTLE LLANO 052 45.0
END DESCRIPTION:
XS GIS Cut Line= 3
      2829355.69     10265653.11      2829061.00     10265706.00
      2829005.65     10265753.14
#Sta/Elev= 30
  4700.6 1155.54  4703.1 1155.54  4727.5 1149.00  4732.5 1148.79  4746.1 1146.74
  4781.2 1141.63  4786.2 1141.53  4792.0 1140.36  4802.2 1139.77  4812.4 1138.36
  4822.5 1137.67  4839.9 1134.69  4845.0 1134.58  4853.0 1133.45  4898.7 1129.53
  4903.8 1129.60  4934.3 1127.59  4952.4 1125.36  4957.5 1125.37  4964.8 1123.98
  5006.4 1119.59  5006.7 1119.09  5010.2 1119.09  5010.4 1119.59  5011.7 1120.46
  5016.1 1123.41  5030.4 1127.57  5037.0 1127.50  5044.7 1128.44  5072.7 1129.97
#Mann=5,-1,0
  4700.6    0.05       0  4746.1    0.12       0  5006.4    0.07       0
  5010.4    0.12       0  5011.7    0.05       0
Bank Sta=5006.4,5010.4
Exp/Cntr=0.3,0.1

Type RM Length L Ch R = 1,22404,476,476,476
BEGIN DESCRIPTION:
LITTLE LLANO 052 44.0
END DESCRIPTION:
XS GIS Cut Line= 3
      2829305.67     10265303.12      2829005.00     10265369.00
      2828855.65     10265403.12
#Sta/Elev= 30
  4692.2 1138.37  4702.2 1137.09  4711.5 1135.57  4743.4 1133.16  4760.5 1132.21
  4765.6 1133.02  4784.3 1131.13  4809.4 1130.38  4907.3 1123.25  4917.4 1116.19
  4925.6 1115.12  4925.9 1114.62  4929.6 1115.12  4937.9 1118.65  4945.0 1120.01
  4946.1 1120.22  4951.2 1115.83  4958.4 1117.31  4968.6 1117.45  4995.0 1115.60
  5002.2 1116.06  5009.6 1118.23  5038.1 1123.41  5043.2 1123.19  5060.8 1126.66
  5081.0 1129.11  5086.1 1128.91  5122.4 1136.35  5134.2 1139.90  5153.2 1142.52
#Mann=5,-1,0
  4692.2    0.05       0  4702.2    0.12       0  4925.6    0.05       0
  4929.6    0.12       0  4945.0    0.05       0
Bank Sta=4925.6,4929.6
Exp/Cntr=0.3,0.1

Type RM Length L Ch R = 1,21928,469,469,469
BEGIN DESCRIPTION:
LITTLE LLANO 052 43.0
END DESCRIPTION:
XS GIS Cut Line= 3
      2829405.70     10265203.13      2829100.00     10264939.00
      2828955.69     10264953.11
#Sta/Elev= 30
  4596.0 1151.82  4599.3 1151.82  4603.2 1150.23  4624.0 1148.94  4638.3 1145.36
  4645.9 1144.39  4660.2 1141.06  4666.8 1140.54  4681.0 1137.12  4709.5 1132.24
  4730.4 1130.08  4752.3 1126.37  4773.2 1124.37  4780.8 1124.83  4794.3 1123.40
  4908.1 1117.51  4971.7 1116.69  4979.3 1115.19  4990.6 1111.50  4990.8 1111.00
  4994.6 1111.50  4999.8 1111.98  5004.7 1111.98  5014.4 1113.65  5054.6 1114.67
  5084.7 1117.46  5091.7 1119.11  5096.7 1118.89  5114.3 1121.60  5145.0 1126.14
#Mann=5,-1,0
  4596.0    0.12       0  4990.6    0.03       0  4994.6    0.12       0
  4999.8    0.05       0  5114.3    0.12       0
Bank Sta=4990.6,4994.6
Exp/Cntr=0.3,0.1

Type RM Length L Ch R = 1,21459,552,552,552
BEGIN DESCRIPTION:
LITTLE LLANO 052 42.0
END DESCRIPTION:
XS GIS Cut Line= 3
      2829505.67     10265003.10      2829251.00     10264680.00
      2828955.70     10264403.12
#Sta/Elev= 30
  4588.6 1131.09  4652.2 1123.74  4695.2 1120.20  4709.6 1118.36  4782.0 1114.59
  4823.5 1113.35  4866.8 1111.06  4873.2 1111.44  4881.3 1110.36  4937.3 1110.96
  4966.2 1109.98  4972.6 1111.24  4987.0 1109.13  4994.8 1106.80  5006.5 1105.84
  5006.7 1105.34  5010.2 1105.34  5010.5 1105.84  5015.8 1106.06  5022.6 1109.51
  5029.9 1110.22  5036.8 1113.23  5044.1 1112.34  5058.3 1114.14  5079.3 1113.65
  5217.9 1115.86  5259.8 1116.78  5320.1 1118.67  5383.6 1122.78  5404.8 1124.80
#Mann=6,-1,0
  4588.6    0.05       0  4782.0    0.12       0  5006.5    0.07       0
  5010.5    0.12       0  5217.9    0.05       0  5259.8    0.12       0
Bank Sta=5006.5,5010.5
Exp/Cntr=0.3,0.1

Type RM Length L Ch R = 1,20907,303,303,303
BEGIN DESCRIPTION:
Mapping XS c731b34f
END DESCRIPTION:
XS GIS Cut Line= 3
      2829722.76     10264993.05      2829707.74     10264632.55
      2829557.53     10264181.93
#Sta/Elev= 30
  4700.9 1124.48  4780.9 1119.16  4813.6 1115.26  4820.9 1114.34  4851.0 1113.39
  4871.0 1111.45  4891.0 1111.24  4951.1 1106.15  4961.1 1104.52  4971.1 1104.88
  4981.1 1102.77  4991.5 1101.74  4991.8 1101.24  4995.5 1101.74  5001.1 1102.11
  5011.1 1105.56  5031.1 1108.87  5103.3 1109.27  5149.0 1110.68  5338.7 1121.62
  5344.8 1122.94  5365.1 1125.29  5377.3 1125.38  5402.0 1127.23  5428.3 1131.21
  5491.6 1136.35  5496.8 1135.78  5523.2 1139.31  5528.5 1138.66  5536.7 1139.67
#Mann=5,-1,0
  4700.9    0.05       0  4813.6    0.12       0  4991.5    0.07       0
  4995.5    0.12       0  5344.8    0.05       0
Bank Sta=4991.5,4995.5
Exp/Cntr=0.3,0.1

Type RM Length L Ch R = 1,20604,428,428,428
BEGIN DESCRIPTION:
LITTLE LLANO 052 40.0
END DESCRIPTION:
XS GIS Cut Line= 3
      2830005.68     10264803.14      2830009.00     10264711.00
      2829905.67     10264403.07
#Sta/Elev= 30
  4907.8 1110.03  4927.8 1108.61  4937.8 1108.25  4967.9 1104.94  4977.9 1104.45
  4996.4 1100.99  5000.0 1100.99  5006.3 1099.20  5006.6 1098.70  5010.1 1098.70
  5010.3 1099.20  5019.2 1099.78  5025.1 1103.22  5030.4 1104.05  5056.7 1105.13
  5071.6 1104.83  5093.5 1105.18  5103.3 1104.59  5113.8 1104.83  5119.8 1104.26
  5134.9 1104.80  5151.3 1104.61  5166.5 1106.02  5214.4 1109.38  5229.8 1109.81
  5245.9 1111.42  5272.0 1112.97  5277.5 1113.71  5305.2 1115.31  5324.8 1116.34
#Mann=5,-1,0
  4907.8    0.05       0  5006.3    0.05       0  5010.3    0.05       0
  5019.2    0.12       0  5305.2    0.05       0
Bank Sta=5006.3,5010.3
Exp/Cntr=0.3,0.1

Type RM Length L Ch R = 1,20176,452,452,452
BEGIN DESCRIPTION:
LITTLE LLANO 052 39.0
END DESCRIPTION:
XS GIS Cut Line= 3
      2830255.69     10264803.14      2830184.75     10264487.00
      2830105.68     10264253.10
#Sta/Elev= 30
  4676.0 1109.85  4727.3 1108.21  4778.5 1105.50  4786.9 1105.86  4879.4 1104.27
  4901.5 1105.01  4952.7 1105.10  4963.0 1103.75  4970.5 1101.16  4975.6 1101.68
  4983.5 1098.72  4991.7 1097.75  4992.0 1097.25  4995.5 1097.25  4995.7 1097.75
  4999.4 1099.43  5004.7 1099.43  5011.0 1101.62  5016.3 1101.61  5042.5 1106.32
  5073.2 1109.44  5105.4 1113.00  5110.7 1112.92  5134.6 1116.81  5168.3 1122.35
  5205.0 1126.53  5225.8 1130.13  5231.2 1132.62  5236.4 1132.13  5246.9 1133.81
#Mann=6,-1,0
  4676.0    0.12       0  4879.4    0.05       0  4991.7    0.05       0
  4995.7    0.05       0  5073.2    0.12       0  5134.6    0.05       0
Bank Sta=4991.7,4995.7
Exp/Cntr=0.3,0.1

Type RM Length L Ch R = 1,19724,494,494,494
BEGIN DESCRIPTION:
LITTLE LLANO 052 38.0
END DESCRIPTION:
XS GIS Cut Line= 3
      2830655.66     10264853.07      2830477.75     10264573.00
      2830755.67     10263953.15
#Sta/Elev= 30
  4668.2 1115.70  4787.5 1108.22  4816.4 1106.69  4869.7 1102.27  4899.9 1101.56
  4921.4 1101.10  4976.9 1095.73  4977.2 1095.23  4981.1 1095.73  5006.3 1096.20
  5052.6 1099.25  5058.1 1100.69  5075.8 1098.86  5081.3 1102.13  5098.5 1100.28
  5120.4 1103.26  5202.7 1102.59  5219.1 1103.97  5231.3 1100.69  5254.5 1098.82
  5311.9 1100.64  5347.2 1101.51  5375.9 1104.39  5399.1 1103.43  5497.3 1110.23
  5536.9 1117.19  5566.8 1126.43  5590.0 1131.29  5624.5 1136.69  5679.3 1142.56
#Mann=7,-1,0
  4668.2    0.05       0  4787.5    0.12       0  4816.4    0.05       0
  4899.9    0.12       0  4976.9    0.07       0  4981.1    0.12       0
  5311.9    0.05       0
Bank Sta=4976.9,4981.1
Exp/Cntr=0.3,0.1

Type RM Length L Ch R = 1,19230,357,357,357
BEGIN DESCRIPTION:
LITTLE LLANO 052 37.0
END DESCRIPTION:
XS GIS Cut Line= 3
      2831255.68     10265153.09      2830880.00     10264353.00
      2830905.69     10264053.10
#Sta/Elev= 30
  4116.1 1166.43  4153.1 1161.70  4227.0 1148.42  4261.4 1143.85  4317.9 1136.44
  4332.8 1134.41  4348.1 1132.11  4381.2 1130.06  4409.5 1124.42  4529.1 1112.00
  4591.1 1104.10  4625.9 1103.29  4688.8 1098.54  4701.6 1099.89  4734.4 1096.79
  4911.5 1098.73  4956.3 1096.09  4973.6 1092.83  4976.9 1090.80  4977.2 1090.30
  4981.2 1090.80  4996.4 1091.07  5006.5 1093.28  5011.5 1091.97  5020.0 1093.43
  5030.0 1097.58  5040.0 1098.85  5130.4 1104.92  5160.5 1108.62  5301.0 1133.94
#Mann=6,-1,0
  4116.1    0.05       0  4261.4    0.12       0  4317.9    0.05       0
  4332.8    0.12       0  4976.9    0.07       0  4981.2    0.12       0
Bank Sta=4976.9,4981.2
Exp/Cntr=0.3,0.1

Type RM Length L Ch R = 1,18873,432,432,432
BEGIN DESCRIPTION:
LITTLE LLANO 052 36.0
END DESCRIPTION:
XS GIS Cut Line= 3
      2831205.68     10264903.11      2831102.75     10264508.00
      2831005.68     10264103.07
#Sta/Elev= 30
  4591.7 1129.25  4609.4 1125.96  4614.5 1126.58  4622.7 1124.05  4634.4 1123.56
  4643.4 1122.31  4649.9 1120.17  4655.0 1120.58  4690.4 1115.75  4788.0 1107.86
  4806.7 1105.38  4870.7 1101.21  4912.0 1095.58  4928.2 1092.05  4953.4 1093.52
  4984.4 1092.11  4994.7 1090.25  4997.8 1087.80  4998.0 1087.30  5002.1 1087.80
  5015.3 1088.14  5025.6 1091.24  5051.5 1093.68  5056.7 1093.07  5093.5 1096.65
  5224.7 1100.93  5323.8 1107.17  5334.1 1109.46  5385.5 1117.14  5416.4 1124.00
#Mann=4,-1,0
  4591.7    0.05       0  4634.4    0.12       0  4997.8    0.07       0
  5002.1    0.12       0
Bank Sta=4997.8,5002.1
Exp/Cntr=0.3,0.1

Type RM Length L Ch R = 1,18441,410,410,410
BEGIN DESCRIPTION:
LITTLE LLANO 052 35.0
END DESCRIPTION:
XS GIS Cut Line= 3
      2831455.69     10264853.07      2831481.50     10264530.00
      2831205.70     10264253.13
#Sta/Elev= 30
  4675.9 1131.06  4706.0 1126.35  4734.8 1120.25  4739.9 1120.55  4746.1 1118.68
  4776.2 1114.73  4816.3 1108.15  4926.7 1097.33  4936.7 1095.91  4956.8 1091.09
  4976.8 1088.80  4985.8 1086.85  4990.8 1087.14  4995.9 1086.26  5006.8 1083.36
  5007.1 1082.86  5011.2 1083.36  5016.1 1084.89  5023.1 1088.63  5037.3 1092.34
  5044.3 1093.33  5079.7 1093.47  5086.8 1094.19  5108.0 1093.61  5256.5 1094.68
  5320.1 1097.87  5334.3 1097.89  5355.5 1099.63  5365.6 1099.56  5390.8 1101.86
#Mann=4,-1,0
  4675.9    0.12       0  5006.8    0.07       0  5011.2    0.12       0
  5365.6    0.05       0
Bank Sta=5006.8,5011.2
Exp/Cntr=0.3,0.1

Type RM Length L Ch R = 1,18031,430,430,430
BEGIN DESCRIPTION:
LITTLE LLANO 052 34.0
END DESCRIPTION:
XS GIS Cut Line= 3
      2831905.68     10264753.10      2831843.50     10264369.00
      2831455.65     10263953.08
#Sta/Elev= 30
  4610.9 1125.72  4681.8 1116.73  4767.6 1107.34  4773.0 1105.91  4854.5 1095.99
  4864.1 1094.86  4935.1 1091.63  4957.2 1089.00  4973.4 1080.71  4973.7 1080.21
  4977.8 1080.71  4985.7 1082.61  5000.0 1083.50  5045.2 1088.93  5059.3 1089.54
  5066.2 1088.58  5080.3 1089.01  5094.5 1090.46  5165.4 1090.48  5236.2 1093.05
  5299.7 1096.88  5342.2 1100.21  5413.1 1107.31  5462.4 1110.72  5490.7 1114.26
  5504.9 1114.88  5526.4 1117.72  5533.2 1119.68  5540.6 1119.92  5568.7 1124.09
#Mann=5,-1,0
  4610.9    0.05       0  4854.5    0.12       0  4957.2    0.05       0
  4973.4    0.05       0  4977.8    0.05       0
Bank Sta=4973.4,4977.8
Exp/Cntr=0.3,0.1

Type RM Length L Ch R = 1,17601,499,499,499
BEGIN DESCRIPTION:
LITTLE LLANO 052 33.0
END DESCRIPTION:
XS GIS Cut Line= 3
      2832055.69     10264553.10      2832234.25     10264253.00
      2832105.69     10263703.13
#Sta/Elev= 30
  4650.8 1100.69  4687.9 1097.91  4732.2 1093.36  4759.8 1092.84  4775.4 1090.27
  4799.4 1088.61  4913.7 1085.01  4929.3 1083.94  4935.1 1082.15  4950.7 1082.88
  4956.5 1079.73  4972.1 1082.13  4977.9 1078.77  4987.7 1080.18  4991.2 1077.76
  4991.6 1077.26  4995.8 1077.76  5020.4 1079.56  5030.7 1081.45  5041.0 1087.32
  5058.0 1089.20  5133.4 1088.92  5195.8 1090.37  5225.8 1091.48  5246.4 1094.55
  5266.9 1093.02  5455.9 1106.94  5533.9 1115.92  5546.0 1119.46  5564.7 1119.69
#Mann=6,-1,0
  4650.8    0.12       0  4687.9    0.05       0  4799.4    0.12       0
  4991.2    0.07       0  4995.8    0.12       0  5020.4    0.05       0
Bank Sta=4991.2,4995.8
Exp/Cntr=0.3,0.1

Type RM Length L Ch R = 1,17102,466,466,466
BEGIN DESCRIPTION:
LITTLE LLANO 052 32.0
END DESCRIPTION:
XS GIS Cut Line= 3
      2832605.68     10264803.11      2832593.50     10264403.00
      2832155.71     10263703.15
#Sta/Elev= 30
  4599.7 1112.83  4629.7 1108.33  4669.7 1103.87  4764.4 1097.93  4886.4 1087.34
  4929.9 1085.19  4979.9 1081.69  4989.9 1080.59  4997.4 1078.30  5002.7 1078.30
  5009.4 1076.40  5009.7 1075.90  5014.0 1076.40  5020.9 1078.44  5042.1 1082.08
  5063.3 1083.52  5252.0 1085.36  5367.5 1088.42  5419.4 1090.66  5440.6 1090.76
  5477.1 1092.63  5492.5 1095.71  5519.6 1094.24  5550.2 1097.67  5650.5 1103.99
  5738.9 1111.58  5781.3 1113.15  5790.2 1112.86  5812.0 1117.38  5825.5 1119.05
#Mann=4,-1,0
  4599.7    0.12       0  4886.4    0.05       0  5009.4    0.03       0
  5014.0    0.05       0
Bank Sta=5009.4,5014
Exp/Cntr=0.3,0.1

Type RM Length L Ch R = 1,16636,402,402,402
BEGIN DESCRIPTION:
LITTLE LLANO 052 31.0
END DESCRIPTION:
XS GIS Cut Line= 3
      2832805.68     10264703.13      2832962.00     10264128.00
      2832905.68     10263703.12
#Sta/Elev= 30
  4404.0 1103.07  4435.1 1101.05  4461.1 1101.33  4476.6 1099.05  4562.5 1090.98
  4600.4 1088.75  4658.9 1085.24  4683.8 1084.12  4735.6 1083.31  4769.1 1083.61
  4797.8 1082.64  4891.1 1082.23  4917.9 1080.61  4923.0 1081.02  4963.6 1079.28
  4984.3 1075.71  5005.0 1075.13  5007.6 1074.43  5008.0 1073.93  5012.0 1073.93
  5012.3 1074.43  5015.0 1074.70  5025.1 1078.74  5035.2 1081.80  5216.8 1088.17
  5277.3 1092.15  5327.7 1094.63  5347.9 1096.62  5368.1 1096.72  5428.6 1100.48
#Mann=6,-1,0
  4404.0    0.12       0  4562.5    0.05       0  4600.4    0.12       0
  4658.9    0.05       0  5007.6    0.05       0  5012.3    0.05       0
Bank Sta=5007.6,5012.3
Exp/Cntr=0.3,0.1

Type RM Length L Ch R = 1,16234,457,457,457
BEGIN DESCRIPTION:
LITTLE LLANO 052 30.0
END DESCRIPTION:
XS GIS Cut Line= 3
      2832805.69     10264853.10      2833343.50     10264110.00
      2833005.69     10263753.12
#Sta/Elev= 30
  4082.7 1103.63  4161.2 1098.86  4226.2 1098.27  4247.0 1096.89  4397.8 1092.92
  4456.7 1088.08  4534.0 1083.03  4560.2 1082.48  4755.9 1081.55  4835.6 1079.85
  4885.1 1077.33  4963.2 1077.65  4971.5 1077.25  4977.9 1073.03  4981.7 1072.13
  4982.1 1071.63  4986.4 1072.13  5038.5 1073.14  5045.8 1074.77  5060.0 1075.37
  5123.5 1074.71  5130.8 1077.38  5137.7 1077.06  5159.1 1080.07  5194.3 1082.48
  5215.7 1082.82  5222.6 1080.75  5236.8 1083.18  5463.3 1094.64  5491.4 1097.44
#Mann=5,-1,0
  4082.7    0.05       0  4456.7    0.12       0  4560.2    0.05       0
  4981.7    0.03       0  4986.4    0.05       0
Bank Sta=4981.7,4986.4
Exp/Cntr=0.3,0.1

Type RM Length L Ch R = 1,15777,477,477,477
BEGIN DESCRIPTION:
LITTLE LLANO 052 29.0
END DESCRIPTION:
XS GIS Cut Line= 3
      2833905.67     10264653.07      2833731.50     10263921.00
      2833655.68     10263703.11
#Sta/Elev= 30
  4247.5 1094.08  4266.0 1092.89  4271.1 1093.58  4288.6 1091.72  4319.4 1090.64
  4432.5 1084.01  4444.9 1084.65  4453.0 1083.51  4504.4 1079.99  4514.7 1080.87
  4545.5 1078.62  4576.5 1078.41  4613.5 1076.51  4668.9 1076.60  4679.2 1075.92
  4740.0 1075.55  4792.4 1076.70  4967.0 1077.19  4977.3 1075.59  4996.3 1070.14
  5000.0 1070.14  5000.4 1069.14  5000.7 1068.64  5005.2 1069.14  5050.7 1074.44
  5071.9 1077.67  5167.2 1085.47  5198.9 1089.26  5228.9 1091.05  5230.7 1091.05
#Mann=4,-1,0
  4247.5    0.05       0  5000.4    0.05       0  5005.2    0.05       0
  5228.9    0.12       0
Bank Sta=5000.4,5005.2
Exp/Cntr=0.3,0.1

Type RM Length L Ch R = 1,15300,486,486,486
BEGIN DESCRIPTION:
LITTLE LLANO 052 28.0
END DESCRIPTION:
XS GIS Cut Line= 3
      2833905.70     10264753.07      2834162.50     10263999.00
      2833955.69     10263653.11
#Sta/Elev= 30
  4203.4 1099.25  4276.7 1095.87  4319.8 1093.40  4478.0 1083.57  4488.6 1084.94
  4496.0 1084.65  4527.3 1080.84  4558.7 1079.49  4573.1 1080.31  4590.0 1078.69
  4636.5 1077.99  4678.7 1075.78  4840.9 1073.12  4974.5 1074.83  4985.1 1070.85
  4992.4 1066.37  4994.8 1066.12  4995.1 1065.62  4999.6 1066.12  5023.7 1066.87
  5039.2 1069.97  5045.1 1068.49  5060.6 1071.70  5066.5 1070.40  5076.2 1072.99
  5082.0 1072.63  5088.4 1074.05  5241.5 1076.95  5368.0 1082.86  5403.0 1083.44
#Mann=5,-1,0
  4203.4    0.05       0  4276.7    0.12       0  4319.8    0.05       0
  4994.8    0.03       0  4999.6    0.05       0
Bank Sta=4994.8,4999.6
Exp/Cntr=0.3,0.1

Type RM Length L Ch R = 1,14814,981,981,981
BEGIN DESCRIPTION:
LITTLE LLANO 052 27.0
END DESCRIPTION:
XS GIS Cut Line= 3
      2834055.66     10264503.13      2834631.25     10264090.00
      2835005.71     10263503.08
#Sta/Elev= 30
  4291.5 1083.34  4319.8 1085.29  4370.1 1080.75  4470.8 1078.41  4592.4 1070.82
  4607.1 1067.56  4672.2 1062.71  4678.3 1065.15  4707.8 1062.84  4713.9 1065.53
  4728.7 1062.42  4734.8 1065.37  4743.4 1063.82  4764.3 1067.55  4850.2 1070.81
  4943.9 1069.49  4965.7 1065.55  4986.5 1065.22  4990.4 1062.07  4990.8 1061.57
  4995.9 1062.07  5015.8 1064.51  5021.8 1069.80  5031.0 1071.07  5088.6 1065.25
  5161.4 1067.74  5188.5 1064.06  5233.5 1073.57  5399.6 1072.86  5696.2 1086.44
#Mann=3,-1,0
  4291.5    0.05       0  4990.4    0.03       0  4995.9    0.05       0
Bank Sta=4990.4,4995.9
Exp/Cntr=0.3,0.1

Type RM Length L Ch R = 1,13833,456,456,456
BEGIN DESCRIPTION:
LITTLE LLANO 052 26.0
END DESCRIPTION:
XS GIS Cut Line= 3
      2834905.68     10264603.09      2834903.50     10264361.00
      2835205.70     10263553.07
#Sta/Elev= 30
  4757.9 1074.74  4807.9 1071.57  4847.9 1065.77  4915.0 1063.93  4977.9 1062.10
  4993.6 1057.44  4994.1 1056.94  4999.2 1057.44  5008.4 1058.13  5029.8 1063.00
  5047.4 1064.21  5157.9 1063.94  5188.2 1063.06  5211.3 1061.19  5218.5 1061.69
  5232.6 1065.57  5273.7 1068.30  5425.1 1067.65  5621.1 1070.73  5659.7 1073.67
  5670.4 1075.49  5676.4 1078.77  5681.7 1076.33  5691.7 1079.23  5701.3 1079.73
  5731.6 1079.56  5736.9 1078.33  5792.2 1081.80  5809.2 1081.95  5862.6 1086.63
#Mann=4,-1,0
  4757.9    0.12       0  4915.0    0.05       0  4993.6    0.03       0
  4999.2    0.05       0
Bank Sta=4993.6,4999.2
Exp/Cntr=0.3,0.1

Type RM Length L Ch R = 1,13377,538,538,538
BEGIN DESCRIPTION:
LITTLE LLANO 052 25.0
END DESCRIPTION:
XS GIS Cut Line= 3
      2835255.67     10264553.14      2835356.50     10264405.00
      2835255.68     10263603.11
#Sta/Elev= 30
  4820.8 1077.65  4864.2 1071.72  4870.3 1072.46  4879.2 1070.78  4885.2 1071.17
  4900.1 1068.57  4921.1 1067.86  4929.0 1066.42  4936.1 1063.91  4942.1 1064.02
  4951.0 1061.89  4965.9 1059.98  5003.5 1056.90  5008.9 1054.91  5009.4 1054.41
  5015.0 1054.91  5032.1 1057.27  5041.9 1059.80  5046.9 1058.73  5052.3 1061.28
  5062.4 1064.41  5082.5 1065.72  5112.8 1064.93  5132.9 1065.59  5253.9 1063.55
  5405.1 1064.58  5515.9 1066.65  5646.9 1071.25  5798.1 1080.94  5808.2 1082.59
#Mann=4,-1,0
  4820.8    0.12       0  4929.0    0.05       0  5008.9    0.05       0
  5015.0    0.05       0
Bank Sta=5008.9,5015
Exp/Cntr=0.3,0.1

Type RM Length L Ch R = 1,12839,408,408,408
BEGIN DESCRIPTION:
Mapping XS 1ec953e6
END DESCRIPTION:
XS GIS Cut Line= 3
      2835761.38     10264677.62      2835791.43     10264287.06
      2835626.45     10263597.13
#Sta/Elev= 30
  4395.8 1077.47  4450.5 1074.50  4500.6 1069.85  4505.9 1070.37  4521.4 1073.67
  4601.1 1073.92  4646.7 1072.27  4651.8 1073.31  4701.2 1072.71  4782.1 1068.90
  4855.5 1063.73  4884.1 1061.52  4919.9 1060.70  4962.0 1053.50  4997.2 1052.31
  5006.0 1050.12  5006.5 1049.62  5012.3 1050.12  5028.1 1053.71  5058.9 1055.79
  5079.5 1060.06  5088.2 1060.74  5151.4 1060.32  5254.3 1061.74  5261.5 1063.09
  5303.6 1064.09  5387.7 1069.41  5408.5 1071.23  5434.9 1076.00  5496.9 1080.11
#Mann=6,-1,0
  4395.8    0.12       0  4505.9    0.05       0  4601.1    0.12       0
  4855.5    0.05       0  5006.0    0.05       0  5012.3    0.05       0
Bank Sta=5006,5012.3
Exp/Cntr=0.3,0.1

Type RM Length L Ch R = 1,12431,472,472,472
BEGIN DESCRIPTION:
LITTLE LLANO 052 23.0
END DESCRIPTION:
XS GIS Cut Line= 3
      2836005.68     10264253.12      2836100.00     10263903.00
      2836355.66     10263503.15
#Sta/Elev= 30
  4637.4 1072.21  4651.8 1070.36  4744.7 1063.81  4793.9 1060.88  4894.5 1057.84
  4906.7 1057.53  4917.0 1056.09  4924.0 1053.68  4963.9 1050.35  4994.2 1048.76
  4994.7 1048.26  5000.6 1048.76  5024.7 1049.36  5034.0 1051.18  5039.9 1050.01
  5047.3 1053.12  5055.1 1054.64  5085.6 1054.03  5106.7 1053.61  5133.8 1051.85
  5185.4 1051.87  5206.5 1050.94  5249.1 1058.90  5264.0 1059.62  5272.9 1058.89
  5285.2 1060.90  5359.7 1066.09  5403.4 1069.33  5424.7 1071.74  5474.6 1075.02
#Mann=9,-1,0
  4637.4    0.05       0  4651.8    0.12       0  4744.7    0.05       0
  4793.9    0.12       0  4894.5    0.05       0  4994.2    0.07       0
  5000.6    0.05       0  5085.6    0.05       0  5359.7    0.12       0
Bank Sta=4994.2,5000.6
Exp/Cntr=0.3,0.1

Type RM Length L Ch R = 1,11959,461,461,461
BEGIN DESCRIPTION:
LITTLE LLANO 052 22.0
END DESCRIPTION:
XS GIS Cut Line= 3
      2836355.69     10264253.10      2836558.50     10263877.00
      2836405.68     10263453.11
#Sta/Elev= 30
  4572.7 1067.59  4602.7 1064.56  4668.4 1061.01  4674.9 1060.05  4726.4 1057.84
  4743.1 1056.65  4772.2 1056.32  4799.9 1054.99  4881.7 1054.98  4911.7 1050.26
  4919.8 1049.40  4963.6 1048.64  4985.5 1047.36  4993.1 1045.99  4996.1 1044.72
  4996.6 1044.22  5002.6 1044.72  5014.8 1045.43  5021.6 1050.49  5026.9 1048.64
  5036.0 1050.85  5128.0 1055.08  5200.4 1058.93  5287.1 1065.51  5323.1 1067.01
  5365.6 1070.66  5379.2 1072.65  5429.3 1075.85  5440.6 1077.53  5450.6 1078.06
#Mann=6,-1,0
  4572.7    0.05       0  4726.4    0.12       0  4911.7    0.05       0
  4996.1    0.05       0  5002.6    0.05       0  5128.0    0.12       0
Bank Sta=4996.1,5002.6
Exp/Cntr=0.3,0.1

Type RM Length L Ch R = 1,11498,499,499,499
BEGIN DESCRIPTION:
LITTLE LLANO 052 21.0
END DESCRIPTION:
XS GIS Cut Line= 3
      2837105.69     10264353.13      2836980.25     10263941.00
      2836705.70     10263553.14
#Sta/Elev= 30
  4569.2 1069.19  4618.5 1064.60  4708.1 1059.18  4778.3 1055.17  4831.3 1053.29
  4893.1 1052.20  4929.8 1051.66  4935.1 1051.00  4962.7 1050.47  4967.9 1050.91
  4976.9 1049.57  4987.3 1046.84  4992.1 1043.16  4992.6 1042.66  4998.4 1042.66
  4998.9 1043.16  5009.7 1043.39  5016.2 1044.53  5045.7 1045.39  5058.7 1047.47
  5081.4 1047.79  5087.5 1048.89  5102.3 1047.06  5117.1 1046.80  5138.0 1047.67
  5173.7 1052.15  5245.1 1052.21  5295.5 1053.66  5426.0 1059.27  5475.2 1062.36
#Mann=5,-1,0
  4569.2    0.05       0  4708.1    0.12       0  4893.1    0.05       0
  4992.1    0.05       0  4998.9    0.05       0
Bank Sta=4992.1,4998.9
Exp/Cntr=0.3,0.1

Type RM Length L Ch R = 1,10999,462,462,462
BEGIN DESCRIPTION:
LITTLE LLANO 052 20.0
END DESCRIPTION:
XS GIS Cut Line= 3
      2837505.66     10264103.07      2837415.25     10263948.00
      2837305.67     10263753.09
#Sta/Elev= 30
  4820.5 1064.11  4849.8 1056.58  4871.3 1055.84  4887.0 1050.88  4901.5 1048.04
  4924.2 1046.49  4951.5 1046.84  4967.3 1045.18  4973.0 1045.69  4981.4 1043.59
  4988.8 1039.85  5006.8 1039.61  5007.3 1039.11  5013.8 1039.61  5026.3 1042.50
  5032.0 1041.42  5040.0 1043.72  5047.9 1044.50  5053.7 1043.40  5063.0 1044.46
  5069.6 1046.47  5075.4 1045.14  5085.6 1047.84  5091.3 1043.99  5097.4 1047.96
  5107.2 1048.65  5113.0 1045.44  5120.3 1048.62  5166.2 1048.39  5223.6 1050.76
#Mann=4,-1,0
  4820.5    0.12       0  4981.4    0.05       0  5006.8    0.03       0
  5013.8    0.05       0
Bank Sta=5006.8,5013.8
Exp/Cntr=0.3,0.1

Type RM Length L Ch R = 1,10537,840,840,840
BEGIN DESCRIPTION:
LITTLE LLANO 052 19.0
END DESCRIPTION:
XS GIS Cut Line= 3
      2837905.68     10264003.10      2837859.25     10263874.00
      2837455.69     10263453.12
#Sta/Elev= 30
  4862.8 1056.21  4878.1 1055.51  4884.0 1053.95  4908.9 1052.06  4958.4 1047.04
  4965.0 1044.22  4979.7 1039.72  4990.3 1038.58  4992.2 1037.77  4992.7 1037.27
  4998.7 1037.27  4999.2 1037.77  5045.5 1043.11  5066.9 1043.30  5123.5 1045.18
  5180.1 1044.53  5201.2 1045.10  5250.6 1044.44  5257.8 1043.97  5286.1 1044.07
  5335.5 1045.64  5349.6 1045.53  5406.2 1049.71  5420.4 1049.93  5448.7 1051.82
  5459.4 1052.05  5552.0 1056.95  5576.0 1059.04  5579.6 1059.95  5583.1 1059.95
#Mann=5,-1,0
  4862.8    0.05       0  4992.2    0.03       0  4999.2    0.05       0
  5459.4    0.12       0  5552.0    0.05       0
Bank Sta=4992.2,4999.2
Exp/Cntr=0.3,0.1

Type RM Length L Ch R = 1,9697,443,443,443
BEGIN DESCRIPTION:
LITTLE LLANO 052 18.0
END DESCRIPTION:
XS GIS Cut Line= 3
      2838055.70     10264053.09      2838488.00     10263372.00
      2838255.72     10263103.15
#Sta/Elev= 30
  4193.3 1057.19  4389.0 1048.00  4461.8 1045.79  4534.7 1044.41  4548.6 1045.40
  4607.5 1042.76  4707.5 1041.12  4795.6 1040.80  4844.7 1042.24  4895.5 1040.99
  4989.6 1036.82  5025.5 1034.02  5026.0 1033.52  5032.6 1034.02  5036.7 1037.38
  5086.1 1040.00  5092.7 1040.58  5100.3 1042.72  5106.9 1041.87  5114.6 1043.53
  5121.2 1042.60  5128.8 1045.03  5135.4 1045.01  5143.1 1047.74  5149.7 1047.72
  5163.9 1043.90  5184.8 1043.30  5199.1 1043.71  5227.6 1047.34  5355.3 1053.21
#Mann=3,-1,0
  4193.3    0.05       0  5025.5    0.03       0  5032.6    0.05       0
Bank Sta=5025.5,5032.6
Exp/Cntr=0.3,0.1

Type RM Length L Ch R = 1,9254,473,473,473
BEGIN DESCRIPTION:
LITTLE LLANO 052 17.0
END DESCRIPTION:
XS GIS Cut Line= 3
      2837955.67     10264203.12      2838759.00     10263642.00
      2838855.68     10263253.14
#Sta/Elev= 30
  4020.1 1065.98  4322.3 1050.38  4400.0 1049.71  4422.7 1048.83  4429.6 1047.72
  4435.7 1048.42  4444.5 1047.54  4465.4 1047.79  4471.5 1047.13  4480.2 1047.97
  4486.3 1046.84  4495.1 1047.37  4501.1 1046.51  4508.0 1046.79  4709.6 1040.56
  4796.0 1039.58  4932.9 1040.25  4968.7 1036.42  4991.4 1032.86  4991.9 1032.36
  4998.5 1032.86  5019.5 1033.50  5088.2 1038.66  5134.6 1038.55  5170.8 1039.72
  5217.3 1038.64  5318.3 1040.68  5359.5 1044.22  5390.4 1048.47  5400.7 1048.68
#Mann=3,-1,0
  4020.1    0.05       0  4991.4    0.03       0  4998.5    0.05       0
Bank Sta=4991.4,4998.5
Exp/Cntr=0.3,0.1

Type RM Length L Ch R = 1,8781,775,775,775
BEGIN DESCRIPTION:
LITTLE LLANO 052 16.0
END DESCRIPTION:
XS GIS Cut Line= 3
      2838355.66     10264403.13      2839160.00     10263892.00
      2839055.68     10262453.08
#Sta/Elev= 30
  4047.0 1049.31  4060.6 1046.79  4438.0 1038.56  4843.1 1036.97  4910.0 1037.83
  4952.4 1034.09  4967.6 1033.74  4990.9 1031.08  4991.4 1030.58  4998.1 1031.08
  5049.0 1033.27  5109.2 1038.90  5131.5 1038.12  5239.5 1038.55  5349.8 1041.04
  5399.9 1040.97  5420.0 1043.27  5440.0 1042.13  5510.2 1041.49  5660.6 1041.94
  5678.8 1042.59  5683.9 1043.75  5770.9 1044.63  5818.2 1044.30  5831.1 1043.18
  5957.5 1043.13  5962.5 1043.99  6231.2 1043.51  6433.2 1046.72  6442.7 1046.89
#Mann=4,-1,0
  4047.0    0.05       0  4990.9    0.03       0  4998.1    0.05       0
  6433.2    0.12       0
Bank Sta=4990.9,4998.1
Exp/Cntr=0.3,0.1

Type RM Length L Ch R = 1,8006,1245,1245,1245
BEGIN DESCRIPTION:
LITTLE LLANO 052 15.0
END DESCRIPTION:
XS GIS Cut Line= 3
      2839655.69     10264553.15      2839637.75     10264467.00
      2839155.69     10263253.12
#Sta/Elev= 30
  4912.0 1043.54  4913.9 1043.54  4932.0 1041.00  4937.1 1041.60  4952.9 1040.00
  4973.3 1036.44  4982.0 1032.30  4987.1 1033.58  4995.6 1027.60  4996.1 1027.10
  5003.3 1027.60  5019.7 1028.51  5025.7 1030.20  5044.0 1032.56  5098.0 1032.54
  5289.7 1036.49  5649.8 1035.77  5751.3 1036.67  5943.0 1036.17  5997.0 1036.83
  6015.6 1036.22  6075.3 1036.46  6123.2 1037.90  6129.3 1037.29  6166.2 1038.59
  6207.6 1038.74  6237.3 1039.84  6252.3 1039.19  6267.0 1040.23  6306.1 1040.57
#Mann=4,-1,0
  4912.0    0.12       0  4913.9    0.05       0  4995.6    0.03       0
  5003.3    0.05       0
Bank Sta=4995.6,5003.3
Exp/Cntr=0.3,0.1

Type RM Length L Ch R = 1,6761,485,485,485
BEGIN DESCRIPTION:
LITTLE LLANO 052 14.0
END DESCRIPTION:
XS GIS Cut Line= 3
      2840005.69     10264453.13      2839708.25     10263739.00
      2839655.69     10263253.14
#Sta/Elev= 30
  4226.4 1051.92  4318.0 1046.13  4341.8 1041.64  4347.2 1036.54  4365.6 1034.00
  4371.1 1028.98  4394.9 1028.79  4400.3 1025.78  4418.7 1029.07  4424.2 1027.04
  4442.6 1029.91  4448.0 1027.22  4471.8 1033.17  4477.2 1033.16  4530.3 1029.63
  4572.6 1031.57  4660.4 1032.18  4891.1 1029.93  5012.1 1023.44  5012.6 1022.94
  5019.8 1023.44  5070.8 1032.13  5217.1 1027.88  5317.7 1027.94  5327.8 1028.18
  5346.1 1031.70  5351.1 1029.54  5368.0 1033.08  5437.8 1038.20  5488.7 1039.83
#Mann=3,-1,0
  4226.4    0.05       0  5012.1    0.05       0  5019.8    0.05       0
Bank Sta=5012.1,5019.8
Exp/Cntr=0.3,0.1

Type RM Length L Ch R = 1,6276,495,495,495
BEGIN DESCRIPTION:
LITTLE LLANO 052 13.0
END DESCRIPTION:
XS GIS Cut Line= 3
      2840055.68     10264353.14      2840148.25     10263571.00
      2840005.70     10263153.15
#Sta/Elev= 30
  4212.4 1048.25  4339.2 1042.20  4454.1 1039.67  4474.2 1038.11  4605.2 1032.33
  4786.4 1029.31  4851.2 1029.17  4887.1 1030.41  4917.3 1029.38  4939.1 1028.11
  4957.6 1024.94  4973.6 1020.96  4974.1 1020.46  4981.8 1020.96  5049.9 1023.06
  5055.1 1024.76  5081.2 1023.75  5086.5 1025.27  5103.4 1024.36  5117.8 1024.69
  5149.1 1022.83  5166.8 1025.40  5188.0 1030.96  5206.5 1034.61  5219.7 1035.35
  5243.1 1034.55  5269.2 1035.69  5325.3 1035.66  5420.4 1038.42  5441.5 1040.09
#Mann=3,-1,0
  4212.4    0.05       0  4973.6    0.05       0  4981.8    0.05       0
Bank Sta=4973.6,4981.8
Exp/Cntr=0.3,0.1

Type RM Length L Ch R = 1,5781,457,457,457
BEGIN DESCRIPTION:
LITTLE LLANO 052 12.0
END DESCRIPTION:
XS GIS Cut Line= 3
      2840255.68     10264103.13      2840568.75     10263469.00
      2840655.70     10263353.09
#Sta/Elev= 30
  4292.8 1038.40  4346.1 1035.71  4374.2 1035.02  4426.6 1031.79  4493.6 1029.46
  4570.6 1028.73  4598.6 1027.71  4688.4 1027.87  4705.3 1027.31  4710.9 1028.03
  4755.8 1026.56  4778.2 1026.31  4783.8 1026.81  4861.6 1025.51  4868.0 1024.43
  4890.4 1022.52  4973.1 1020.53  4994.9 1017.89  4998.0 1016.98  4998.5 1016.48
  5005.9 1016.48  5006.4 1016.98  5023.0 1019.45  5037.6 1023.07  5052.2 1023.17
  5069.6 1025.27  5087.6 1026.77  5102.2 1029.12  5123.0 1031.29  5144.9 1033.09
#Mann=4,-1,0
  4292.8    0.05       0  4998.0    0.03       0  5006.4    0.05       0
  5069.6    0.12       0
Bank Sta=4998,5006.4
Exp/Cntr=0.3,0.1

Type RM Length L Ch R = 1,5324,443,443,443
BEGIN DESCRIPTION:
LITTLE LLANO 052 11.0
END DESCRIPTION:
XS GIS Cut Line= 3
      2840205.68     10264203.11      2841005.00     10263580.00
      2841005.68     10263303.10
#Sta/Elev= 30
  3986.5 1041.24  4100.6 1037.04  4371.0 1028.85  4584.5 1026.79  4692.1 1024.19
  4721.1 1025.07  4727.4 1025.93  4741.9 1025.45  4762.7 1026.53  4876.7 1024.23
  4905.6 1023.46  4934.6 1021.48  4955.4 1018.39  4969.9 1021.30  4976.2 1017.35
  4984.3 1017.20  4990.7 1015.62  5002.6 1015.44  5003.1 1014.94  5010.6 1014.94
  5011.1 1015.44  5016.9 1017.07  5036.9 1019.04  5046.9 1019.17  5076.9 1021.45
  5086.9 1021.33  5126.9 1024.39  5166.9 1028.79  5216.9 1032.02  5276.9 1037.07
#Mann=3,-1,0
  3986.5    0.05       0  5002.6    0.03       0  5011.1    0.05       0
Bank Sta=5002.6,5011.1
Exp/Cntr=0.3,0.1

Type RM Length L Ch R = 1,4881,475,475,475
BEGIN DESCRIPTION:
LITTLE LLANO 052 10.0
END DESCRIPTION:
XS GIS Cut Line= 3
      2841255.69     10264353.11      2841445.00     10263534.00
      2841355.67     10263303.08
#Sta/Elev= 30
  4159.3 1034.75  4220.8 1030.16  4292.7 1026.64  4456.9 1022.38  4492.6 1022.82
  4498.0 1024.30  4528.8 1023.63  4682.7 1023.64  4744.3 1024.76  4867.5 1024.37
  4908.5 1025.23  4929.1 1024.25  4949.6 1022.14  4959.9 1020.23  4970.1 1016.74
  4973.8 1014.61  4974.3 1014.11  4982.3 1014.61  5003.2 1015.48  5022.4 1017.89
  5063.7 1019.52  5086.7 1021.72  5118.2 1023.24  5123.5 1022.79  5148.1 1025.01
  5153.5 1024.55  5183.4 1027.11  5194.0 1029.04  5226.1 1030.43  5247.6 1032.26
#Mann=3,-1,0
  4159.3    0.05       0  4973.8    0.05       0  4982.3    0.05       0
Bank Sta=4973.8,4982.3
Exp/Cntr=0.3,0.1

Type RM Length L Ch R = 1,4406,583,583,583
BEGIN DESCRIPTION:
LITTLE LLANO 052 9.0
END DESCRIPTION:
XS GIS Cut Line= 3
      2842105.67     10264103.06      2841908.75     10263428.00
      2841355.71     10263003.13
#Sta/Elev= 30
  4296.8 1032.35  4335.1 1030.41  4385.7 1026.52  4463.4 1023.06  4646.0 1017.38
  4669.1 1016.71  4741.3 1021.31  4818.7 1019.26  4869.7 1020.34  4885.6 1018.47
  4963.4 1016.96  4984.3 1015.30  4991.3 1013.08  5009.0 1012.42  5009.5 1011.92
  5017.5 1012.42  5019.5 1013.55  5027.7 1014.61  5034.0 1017.07  5048.5 1017.08
  5054.8 1019.81  5063.0 1019.67  5069.3 1021.44  5155.2 1021.25  5470.0 1029.19
  5497.1 1028.04  5519.8 1029.34  5576.0 1028.03  5590.5 1029.44  5697.4 1030.57
#Mann=5,-1,0
  4296.8    0.05       0  4335.1    0.12       0  4646.0    0.05       0
  5009.0    0.03       0  5017.5    0.05       0
Bank Sta=5009,5017.5
Exp/Cntr=0.3,0.1

Type RM Length L Ch R = 1,3823,193,193,193
BEGIN DESCRIPTION:
LITTLE LLANO 052 8.0
END DESCRIPTION:
XS GIS Cut Line= 3
      2842561.64     10263719.05      2842356.41     10263441.38
      2841555.69     10262653.12
#Sta/Elev= 30
  4741.8 1035.59  4774.9 1035.51  4793.3 1036.53  4864.3 1035.48  4878.9 1033.68
  4901.0 1028.50  4914.4 1024.89  4922.8 1023.75  4943.6 1016.73  4979.1 1014.23
  4993.7 1010.91  5010.2 1010.41  5010.7 1009.91  5019.0 1010.41  5029.2 1013.52
  5043.8 1015.10  5079.3 1015.30  5114.7 1017.16  5121.7 1018.47  5135.9 1019.42
  5178.3 1020.33  5454.0 1018.71  5722.8 1019.03  5934.9 1021.40  6041.0 1023.81
  6055.2 1024.46  6069.3 1026.30  6083.5 1024.86  6111.7 1026.99  6210.7 1033.47
#Mann=6,-1,0
  4741.8    0.05       0  4774.9    0.12       0  4901.0    0.05       0
  5010.2    0.05       0  5019.0    0.05       0  6111.7    0.12       0
Bank Sta=5010.2,5019
Exp/Cntr=0.3,0.1

Type RM Length L Ch R = 1,3630,371,371,371
BEGIN DESCRIPTION:
LITTLE LLANO 052 7.0
END DESCRIPTION:
XS GIS Cut Line= 3
      2842655.71     10263503.14      2842578.00     10263420.00
      2841555.68     10262603.11
#Sta/Elev= 30
  4886.2 1034.95  4914.3 1031.56  4928.5 1028.73  4942.7 1022.98  4950.0 1018.69
  4956.8 1016.49  4985.2 1012.82  4991.7 1010.73  5009.8 1009.84  5010.3 1009.34
  5018.6 1009.84  5020.6 1011.14  5035.0 1013.68  5055.8 1014.83  5119.9 1014.97
  5169.5 1020.27  5454.5 1017.71  5917.2 1020.13  6002.0 1022.71  6074.1 1023.54
  6102.9 1025.84  6109.3 1027.56  6123.7 1025.38  6138.1 1025.71  6199.0 1030.06
  6214.9 1031.31  6258.2 1035.18  6272.6 1034.80  6287.0 1037.15  6308.6 1036.64
#Mann=6,-1,0
  4886.2    0.12       0  4991.7    0.05       0  5009.8    0.05       0
  5018.6    0.05       0  6199.0    0.12       0  6214.9    0.05       0
Bank Sta=5009.8,5018.6
Exp/Cntr=0.3,0.1

Type RM Length L Ch R = 1,3259,796,796,796
BEGIN DESCRIPTION:
LITTLE LLANO 052 6.0
END DESCRIPTION:
XS GIS Cut Line= 4
      2843137.22     10263320.68      2842964.13     10263131.49
      2842417.38     10263120.29      2841605.70     10262553.12
#Sta/Elev= 30
  4565.5 1028.61  4664.0 1025.81  4737.7 1025.30  4880.4 1027.27  4940.4 1025.80
  4960.4 1023.21  4970.4 1023.63  4980.4 1016.49  4986.0 1008.85  4996.0 1008.21
  4996.5 1007.71  5004.8 1008.21  5020.4 1011.87  5050.4 1014.37  5180.5 1018.04
  5270.5 1017.31  5367.1 1018.32  5461.1 1015.92  5547.5 1017.93  5598.1 1016.69
  5755.9 1018.50  5834.4 1018.12  5949.5 1019.76  6086.5 1024.54  6128.3 1027.26
  6151.6 1025.79  6209.0 1029.14  6259.2 1031.88  6324.3 1037.63  6359.0 1040.36
#Mann=6,-1,0
  4565.5    0.12       0  4737.7    0.05       0  4996.0    0.03       0
  5004.8    0.05       0  6209.0    0.12       0  6324.3    0.05       0
Bank Sta=4996,5004.8
Exp/Cntr=0.3,0.1

Type RM Length L Ch R = 1,2463,403,403,403
BEGIN DESCRIPTION:
Mapping XS 1b2ec0c3
END DESCRIPTION:
XS GIS Cut Line= 4
      2842875.58     10262974.51      2842646.18     10262749.14
      2842143.10     10262781.34      2841635.99     10262499.62
#Sta/Elev= 30
  4371.5 1026.46  4520.9 1022.44  4527.9 1021.17  4641.1 1016.46  4813.8 1017.00
  4863.9 1015.94  4944.1 1012.27  4964.1 1009.10  4984.2 1007.77  4989.6 1006.05
  4994.6 1006.63  4999.7 1005.15  5000.2 1004.65  5008.7 1005.15  5014.2 1005.58
  5024.3 1008.75  5034.3 1013.99  5044.3 1016.62  5054.3 1017.54  5267.1 1017.13
  5348.3 1018.90  5445.6 1022.74  5489.0 1025.27  5510.8 1028.35  5516.5 1026.41
  5526.0 1025.40  5548.5 1027.89  5619.4 1031.56  5635.5 1031.36  5777.3 1041.24
#Mann=3,-1,0
  4371.5    0.05       0  4999.7    0.05       0  5008.7    0.05       0
Bank Sta=4999.7,5008.7
Exp/Cntr=0.3,0.1

Type RM Length L Ch R = 1,2060,467,467,467
BEGIN DESCRIPTION:
LITTLE LLANO 052 5.0
END DESCRIPTION:
XS GIS Cut Line= 3
      2842815.22     10262817.56      2842655.68     10262503.11
      2842094.81     10262161.55
#Sta/Elev= 30
  4516.1 1019.62  4554.7 1018.01  4593.2 1015.50  4622.0 1014.73  4743.4 1014.46
  4823.9 1015.39  4876.4 1015.14  4913.2 1012.96  4940.4 1010.10  4962.4 1009.96
  4971.3 1009.17  4977.2 1007.02  4985.8 1005.17  4988.2 1003.13  4988.7 1002.63
  4996.7 1002.63  4997.2 1003.13  4998.5 1003.53  5008.1 1003.37  5014.0 1004.25
  5020.9 1007.32  5029.4 1009.65  5050.8 1013.92  5056.6 1014.65  5087.6 1015.85
  5130.2 1014.65  5209.6 1014.61  5393.6 1016.76  5494.3 1018.96  5525.4 1020.10
#Mann=3,-1,0
  4516.1    0.05       0  4988.2    0.03       0  4997.2    0.05       0
Bank Sta=4988.2,4997.2
Exp/Cntr=0.3,0.1

Type RM Length L Ch R = 1,1593,416,416,416
BEGIN DESCRIPTION:
LITTLE LLANO 052 4.0
END DESCRIPTION:
XS GIS Cut Line= 4
      2842891.68     10262970.47      2842823.27     10262286.31
      2842903.99     10262004.81      2843140.94     10261771.43
#Sta/Elev= 30
  4142.2 1026.57  4199.8 1025.57  4322.2 1018.33  4360.6 1015.17  4420.9 1013.26
  4822.9 1013.83  4891.6 1014.99  4925.4 1013.36  4930.6 1011.15  4947.5 1013.08
  4957.9 1012.30  4978.7 1006.14  4989.1 1004.53  5020.4 1002.91  5026.0 1001.91
  5026.5 1001.41  5035.5 1001.91  5037.0 1003.49  5062.0 1006.61  5076.0 1012.58
  5082.8 1018.25  5088.6 1018.87  5127.3 1021.17  5160.4 1027.34  5174.5 1027.84
  5181.5 1026.73  5216.9 1028.96  5278.2 1029.45  5323.0 1028.74  5455.2 1030.37
#Mann=6,-1,0
  4142.2    0.12       0  4322.2    0.05       0  5026.0    0.05       0
  5035.5    0.05       0  5088.6    0.12       0  5278.2    0.05       0
Bank Sta=5026,5035.5
Exp/Cntr=0.3,0.1

Type RM Length L Ch R = 1,1177,396,396,396
BEGIN DESCRIPTION:
LITTLE LLANO 052 3.0
END DESCRIPTION:
XS GIS Cut Line= 3
      2843076.82     10262793.44      2843165.36     10262221.91
      2843253.61     10261876.97
#Sta/Elev= 30
  4644.6 1017.54  4672.4 1014.43  4685.4 1013.22  4738.1 1011.75  4869.2 1012.24
  4908.0 1011.58  4948.5 1012.93  4958.6 1011.35  4968.8 1007.47  4978.9 1001.20
  4989.0  999.69  4995.2 1000.14  5004.4  998.58  5004.9  998.08  5013.5  998.08
  5014.0  998.58  5029.5 1001.09  5049.7 1002.55  5080.1 1006.22  5110.4 1007.44
  5126.3 1009.12  5199.2 1011.30  5232.0 1013.92  5252.7 1016.93  5286.8 1019.39
  5399.4 1024.61  5450.1 1025.47  5526.5 1028.04  5572.7 1028.45  5579.0 1029.32
#Mann=6,-1,0
  4644.6    0.12       0  4672.4    0.05       0  5004.4    0.03       0
  5014.0    0.05       0  5199.2    0.12       0  5399.4    0.05       0
Bank Sta=5004.4,5014
Exp/Cntr=0.3,0.1
