HEC-RAS study LITTLE LLANO RIVER.prj: LITTLE LLANO RIVER Base Level Engineering

--- LITTLE LLANO RIVER.g01 (geometry) --- (continued)

Type RM Length L Ch R = 1 ,42195   ,587,587,587
BEGIN DESCRIPTION:
LITTLE LLANO RIVER 77.0
END DESCRIPTION:
XS GIS Cut Line= 3
      2839955.67     10283253.13      2839727.75       10283489.
      2839405.67     10283803.13
#Sta/Elev= 30
    4672 1107.79  4735.6 1098.48  4756.7 1093.85  4763.9 1093.06  4770.9    1091
    4785 1089.18  4813.3 1087.37  4820.5 1087.78  4955.2 1084.48  4976.2 1083.97
  4996.6 1077.16  4997.1 1076.66  5026.3 1077.16  5032.6 1078.16  5046.7 1077.77
    5075 1080.94  5096.3 1081.21  5121.6 1082.85  5138.8 1083.51  5188.2 1081.13
  5244.8 1084.07  5265.6 1086.12  5273.1 1086.25  5315.5  1092.1    5351 1093.61
  5365.1 1095.63  5386.2 1096.49  5428.7 1100.89  5435.8 1100.55  5449.9 1101.63
#Mann= 6 ,-1 , 0
    4672     .12       0  4955.2     .05       0  4996.6     .05       0
  5026.3     .05       0  5121.6     .12       0  5265.6     .05       0
Bank Sta=4996.6,5026.3
XS Rating Curve= 0 ,0
Exp/Cntr=0.3,0.1

Type RM Length L Ch R = 1 ,41608   ,591,591,591
BEGIN DESCRIPTION:
LITTLE LLANO RIVER 76.0
END DESCRIPTION:
XS GIS Cut Line= 3
      2840005.73     10283103.13      2839600.25       10282968.
      2839255.67      10282753.1
#Sta/Elev= 30
  4572.6 1111.34  4583.2 1111.05    4619 1104.15  4646.4 1100.68  4688.6  1091.3
  4798.3 1084.15  4846.7 1083.35  4873.1 1080.39  4899.4 1079.89  4936.3 1075.44
  4983.7 1073.12  4984.7 1071.16  4985.2 1070.66  5014.5 1071.16  5026.4 1071.73
  5042.1 1071.82  5057.4 1074.45  5072.8 1081.34  5078.7 1080.62    5094 1085.22
  5123.2 1085.26  5188.4 1088.96  5198.6 1088.54  5209.2 1088.49    5225 1090.04
  5230.9 1088.45  5240.3  1090.6  5267.5 1092.77  5377.2 1110.75  5406.1  1112.3
#Mann= 8 ,-1 , 0
  4572.6     .05       0    4619     .12       0  4798.3     .05       0
  4984.7     .05       0  5014.5     .05       0  5026.4     .12       0
  5198.6     .05       0  5209.2     .12       0
Bank Sta=4984.7,5014.5
XS Rating Curve= 0 ,0
Exp/Cntr=0.3,0.1

Type RM Length L Ch R = 1 ,41017   ,511,511,511
BEGIN DESCRIPTION:
Mapping XS b80c3cfd
END DESCRIPTION:
XS GIS Cut Line= 4
      2841208.49     10282826.59      2840514.08     10282652.99
      2839646.02     10282479.38      2839255.38     10282566.19
#Sta/Elev= 30
  3708.7 1115.95  3806.3 1115.25  3876.5 1115.49    3984 1110.56  4034.3 1104.13
  4165.1  1094.9  4235.3 1091.08  4405.7 1086.75  4444.1 1085.84  4473.8 1081.41
  4499.8 1083.78  4568.3 1084.53  4682.4 1083.12  4749.2 1080.58  4761.1 1078.37
  4856.8 1075.61  4912.9 1069.45  4989.2 1066.94  4989.7 1066.44  5019.1 1066.94
  5024.5 1068.79  5136.7 1075.76  5167.8 1080.31  5241.1 1084.26  5299.9 1087.57
  5361.3 1093.91    5474 1096.87  5531.3 1100.47  5660.1 1108.09  5709.9 1111.03
#Mann= 13 ,-1 , 0
  3708.7     .12       0  3806.3     .05       0    3984     .12       0
  4405.7     .05       0  4444.1     .12       0  4568.3     .05       0
  4682.4     .12       0  4761.1     .05       0  4989.2     .03       0
  5019.1     .05       0  5241.1     .12       0  5531.3     .05       0
  5660.1     .12       0
Bank Sta=4989.2,5019.1
XS Rating Curve= 0 ,0
Exp/Cntr=0.3,0.1

Type RM Length L Ch R = 1 ,40506   ,531,531,531
BEGIN DESCRIPTION:
Mapping XS cc0999e5
END DESCRIPTION:
XS GIS Cut Line= 4
      2841165.12     10282783.19      2840579.18     10282414.27
      2840058.35     10282240.66      2839363.91     10282284.06
#Sta/Elev= 30
  4147.4 1113.68  4247.4 1111.56    4328  1107.2  4406.8 1099.41  4629.6 1089.46
  4792.9 1079.83  4838.9 1072.27  4941.9  1067.4    4996 1066.26  5002.5  1065.8
    5003  1065.3  5032.4  1065.8  5039.6 1066.05  5075.4 1067.04  5117.6 1075.58
  5328.4  1083.5  5365.3 1087.68  5450.1 1087.14  5581.8    1089  5621.9 1097.69
    5652 1096.58  5722.1 1100.26  5812.3 1098.41  5862.4 1094.34  5902.5 1097.85
  5942.6 1096.43  5982.6  1098.8  6002.7 1096.15  6022.7 1099.08  6084.6 1099.09
#Mann= 10 ,-1 , 0
  4147.4     .12       0  4247.4     .05       0    4328     .12       0
  4629.6     .05       0  4941.9     .12       0    4996     .05       0
  5002.5     .05       0  5032.4     .05       0  5039.6     .12       0
  5450.1     .05       0
Bank Sta=5002.5,5032.4
XS Rating Curve= 0 ,0
Exp/Cntr=0.3,0.1

Type RM Length L Ch R = 1 ,39975   ,566,566,566
BEGIN DESCRIPTION:
LITTLE LLANO RIVER 73.0
END DESCRIPTION:
XS GIS Cut Line= 3
      2840855.68     10282453.11      2840843.25       10282038.
      2840055.69     10281753.11
#Sta/Elev= 30
  4584.7 1092.13  4604.7 1091.51  4614.7 1089.14  4624.7 1081.79  4644.7 1082.23
  4654.7 1083.99  4664.7 1089.21  4690.2  1088.3  4784.8 1082.71  4864.8 1072.71
  4904.8 1069.56  4934.9 1064.03  4984.9 1062.35    4985 1061.46  4985.5 1060.96
  5014.9 1061.46  5050.6 1063.98  5087.8 1073.43  5113.2 1076.25  5210.4 1080.18
  5316.4 1082.75  5410.4 1086.89  5439.7 1088.51    5465 1088.79  5475.9 1091.13
  5495.7 1090.94  5635.5 1097.36  5699.3 1102.16  5741.8 1107.82  5837.5 1114.52
#Mann= 5 ,-1 , 0
  4584.7     .05       0  4690.2     .12       0    4985     .07       0
  5014.9     .12       0  5410.4     .05       0
Bank Sta=4985,5014.9
XS Rating Curve= 0 ,0
Exp/Cntr=0.3,0.1

Type RM Length L Ch R = 1 ,39409   ,561,561,561
BEGIN DESCRIPTION:
LITTLE LLANO RIVER 72.0
END DESCRIPTION:
XS GIS Cut Line= 3
      2842055.72     10282003.12        2841333.       10281756.
      2840705.73     10281353.14
#Sta/Elev= 30
  4236.2 1103.86    4270 1101.91  4408.4 1090.16    4471 1083.13  4648.3 1071.41
  4677.9 1066.46  4684.9  1065.1  4701.2 1069.58  4726.2 1072.76  4751.8 1075.17
  4778.8 1075.53  4867.5 1071.42  4918.6 1065.11  4954.9 1061.87  4966.7 1059.65
  4992.7 1058.97  4993.7 1057.67  4994.2 1057.17  5023.7 1057.67  5038.7  1058.8
  5050.9 1061.26  5056.9 1065.25  5066.1 1068.18  5093.2 1072.63  5196.3 1076.24
  5347.2 1079.12  5471.7 1083.87  5543.9 1088.34    5627 1093.96  5745.5 1104.55
#Mann= 12 ,-1 , 0
  4236.2     .12       0    4270     .05       0  4677.9     .12       0
  4726.2     .05       0  4751.8     .12       0  4918.6     .05       0
  4993.7     .05       0  5023.7     .05       0  5038.7     .12       0
  5347.2     .05       0  5543.9     .12       0    5627     .05       0
Bank Sta=4993.7,5023.7
XS Rating Curve= 0 ,0
Exp/Cntr=0.3,0.1

Type RM Length L Ch R = 1 ,38848   ,495,495,495
BEGIN DESCRIPTION:
LITTLE LLANO RIVER 71.0
END DESCRIPTION:
XS GIS Cut Line= 3
      2842155.66     10281803.09      2841839.75       10281517.
      2841155.71     10281103.13
#Sta/Elev= 30
  4573.8 1110.87  4609.3 1108.83  4680.2 1099.86  4694.4 1099.99  4757.9 1090.11
  4778.9 1087.97  4814.7 1081.12  4842.2 1078.19    4864 1075.36    4885 1074.36
  4913.4  1067.4  4970.2 1057.98  4991.8 1055.92  5005.3 1055.89  5013.1 1054.15
  5013.6 1053.65  5043.2 1054.15  5056.6 1062.87  5063.2 1064.88  5072.1 1065.88
  5077.9 1068.42  5099.3 1072.19  5114.8 1073.21  5136.1 1072.67  5273.9 1075.89
  5516.3 1075.11  5603.6 1077.81  5647.6 1079.62  5727.7 1087.93  5799.5 1092.85
#Mann= 5 ,-1 , 0
  4573.8     .12       0  4842.2     .05       0  5013.1     .05       0
  5043.2     .05       0  5603.6     .12       0
Bank Sta=5013.1,5043.2
XS Rating Curve= 0 ,0
Exp/Cntr=0.3,0.1

Type RM Length L Ch R = 1 ,38353   ,418,418,418
BEGIN DESCRIPTION:
Mapping XS 00b06fb3
END DESCRIPTION:
XS GIS Cut Line= 3
      2842423.82     10281850.08      2842206.79     10281155.59
      2841186.79     10280830.06
#Sta/Elev= 30
  4329.3 1112.28  4483.3 1114.66  4578.6 1108.52  4638.4 1106.36  4682.3 1102.02
  4708.6 1102.37  4778.8 1097.86    4806 1098.62    4850    1093  4870.9 1091.82
  4881.4 1087.93  4908.7 1082.42  4933.8  1073.9  4941.1 1070.19  4963.8 1051.44
  4964.3 1050.94  4993.9 1051.44  4996.6 1053.38  5017.6 1054.01  5043.8 1057.04
  5055.6  1061.1  5082.9 1065.37  5089.6 1067.82  5109.9 1070.06  5276.1  1073.8
  5742.5 1074.16  5806.9 1075.81  5867.2 1079.19  5969.5 1086.36  6127.6 1090.92
#Mann= 5 ,-1 , 0
  4329.3     .12       0  4963.8     .05       0  4993.9     .12       0
  5867.2     .12       0  5969.5     .05       0
Bank Sta=4963.8,4993.9
XS Rating Curve= 0 ,0
Exp/Cntr=0.3,0.1

Type RM Length L Ch R = 1 ,37935   ,597,597,597
BEGIN DESCRIPTION:
LITTLE LLANO RIVER 69.0
END DESCRIPTION:
XS GIS Cut Line= 3
      2842555.68     10281303.09      2842485.75       10280885.
      2841755.69     10280653.11
#Sta/Elev= 30
  4576.1 1107.78  4656.3 1106.99  4738.3 1104.49  4778.9  1100.7  4791.2 1098.16
  4809.3 1097.58  4839.7 1093.73  4846.8 1091.89  4870.1 1083.46  4900.5 1074.72
  4907.5 1071.68  4912.6 1066.31  4920.8 1063.17  4941.1 1057.38  4961.4 1053.17
  4968.3 1050.75  5002.7 1051.48  5004.2 1049.93  5004.7 1049.43  5034.3 1049.93
    5042 1055.52    5063 1060.75  5083.8  1064.5  5094.5 1068.24    5105 1069.79
  5223.3 1071.76  5314.8 1070.76  5535.2  1072.9  5598.1 1072.66    5766 1076.58
#Mann= 4 ,-1 , 0
  4576.1     .05       0  4656.3     .12       0  5004.2     .07       0
  5034.3     .05       0
Bank Sta=5004.2,5034.3
XS Rating Curve= 0 ,0
Exp/Cntr=0.3,0.1

Type RM Length L Ch R = 1 ,37338   ,453,453,453
BEGIN DESCRIPTION:
LITTLE LLANO RIVER 68.0
END DESCRIPTION:
XS GIS Cut Line= 3
      2842955.68      10280753.1        2842785.       10280370.
      2841805.67     10280553.11
#Sta/Elev= 30
  4580.6  1085.4  4646.9 1086.43  4711.1 1080.65  4716.6  1078.8  4739.8 1077.81
  4768.5 1073.48  4838.2 1077.27  4843.7 1075.66  4861.5 1076.61  4866.9 1074.28
  4884.7  1075.1  4890.2 1071.24  4898.1 1070.84  4907.9 1067.75  4913.4 1063.77
    4920 1061.71  4942.1  1056.6  4974.7 1051.77  4980.5 1048.94    4981 1048.44
  5010.7 1048.94  5029.8 1050.82  5039.5  1049.7  5060.3 1052.37  5090.9  1059.8
  5111.2 1062.19  5149.9 1071.88  5457.1  1069.4  5762.3 1072.09  5996.3 1076.83
#Mann= 3 ,-1 , 0
  4580.6     .12       0  4980.5     .05       0  5010.7     .05       0
Bank Sta=4980.5,5010.7
XS Rating Curve= 0 ,0
Exp/Cntr=0.3,0.1

Type RM Length L Ch R = 1 ,36885   ,577,577,577
BEGIN DESCRIPTION:
LITTLE LLANO RIVER 67.0
END DESCRIPTION:
XS GIS Cut Line= 3
      2843205.71     10280203.14       2842894.5       10279933.
      2841455.68     10278653.11
#Sta/Elev= 30
  4587.9 1074.84  4658.7 1071.93  4701.4 1066.25  4736.5 1065.16  4779.3 1059.31
  4793.5  1055.3  4800.2 1055.51  4807.8 1060.44  4814.4 1058.16  4850.5  1069.6
  4892.5 1067.24  4920.8 1062.01  4977.8 1052.27  4985.2 1048.79  5002.6 1048.37
    5084 1050.81  5133.6 1064.56  5204.4 1069.39  5247.1 1066.39  5388.4 1067.59
  5594.1 1064.15  5657.6 1053.86  5671.1 1047.61  5701.6 1048.11  5785.6 1062.27
    5870 1068.59  6190.6 1065.91  6445.2 1078.97    6600 1093.58  6925.7 1109.22
#Mann= 6 ,-1 , 0
  4587.9     .12       0  4920.8     .05       0  5133.6     .05       0
  5701.6     .05       0  6190.6     .12       0  6445.2     .05       0
Bank Sta=4920.8,5133.6
XS Rating Curve= 0 ,0
Exp/Cntr=0.3,0.1

Type RM Length L Ch R = 1 ,36308   ,547,547,547
BEGIN DESCRIPTION:
LITTLE LLANO RIVER 66.0
END DESCRIPTION:
XS GIS Cut Line= 3
      2843255.71     10279653.13      2842964.75       10279362.
      2841355.73     10278503.13
#Sta/Elev= 30
  4588.4 1070.77  4878.3 1063.33  4913.7 1058.38  4963.2  1056.3  4970.3 1048.48
  4977.3 1049.05  4984.4 1045.21  5012.1 1045.66  5028.4 1049.75  5138.2 1048.74
  5258.5 1064.32  5346.4 1066.03  5384.3 1062.79  5390.3 1055.22  5395.9 1052.66
  5396.7  1044.5  5397.2    1044  5427.7  1044.5  5463.7 1053.03  5598.5 1061.85
  5730.2 1064.31  5973.8 1063.45    6074 1066.49  6183.5 1072.14  6327.9 1081.35
  6415.9 1091.73  6453.9 1093.35  6492.2 1099.54  6667.8 1113.72  6823.9 1119.75
#Mann= 6 ,-1 , 0
  4588.4     .12       0  4963.2     .05       0  5028.4     .05       0
  5427.7     .05       0    6074     .12       0  6183.5     .05       0
Bank Sta=4963.2,5028.4
XS Rating Curve= 0 ,0
Exp/Cntr=0.3,0.1

Type RM Length L Ch R = 1 ,35761   ,599,599,599
BEGIN DESCRIPTION:
LITTLE LLANO RIVER 65.0
END DESCRIPTION:
XS GIS Cut Line= 3
      2843655.65     10278753.12       2842888.5       10278826.
      2842355.69     10278353.11
#Sta/Elev= 30
  4229.4 1085.23    4255 1083.62  4349.9 1073.23  4400.1 1069.47  4470.4 1065.99
  4567.4 1065.37  4681.9 1064.52    4822 1061.56  4842.1 1060.76  4881.1 1056.67
    4912 1050.65    4917 1051.04  4922.5 1048.58  4932.5  1046.7  4982.7 1047.88
  5032.1 1046.43    5068 1048.49  5174.2  1044.3  5188.5 1045.85  5195.1 1045.33
  5201.4 1042.39  5201.9 1041.89  5232.5 1042.39  5244.5 1042.43  5280.5 1052.63
  5323.1 1060.61  5379.1    1064  5451.3 1064.74  5611.5 1070.73  5712.4 1074.94
#Mann= 9 ,-1 , 0
  4229.4     .05       0    4255     .12       0  4567.4     .05       0
  4681.9     .12       0  4881.1     .05       0  5201.4     .05       0
  5232.5     .05       0  5451.3     .12       0  5611.5     .05       0
Bank Sta=5201.4,5232.5
XS Rating Curve= 0 ,0
Exp/Cntr=0.3,0.1

Type RM Length L Ch R = 1 ,35162   ,436,436,436
BEGIN DESCRIPTION:
LITTLE LLANO RIVER 64.0
END DESCRIPTION:
XS GIS Cut Line= 3
       2843655.7     10278703.12      2842877.75       10278231.
      2842505.69     10278053.11
#Sta/Elev= 30
    4090 1084.11  4099.9 1082.85  4125.1 1079.99  4214.1 1072.91    4326 1066.44
  4394.4  1064.4  4578.5 1063.66  4642.5 1061.83    4722 1061.05  4774.3 1056.83
  4811.1 1051.62  4890.6 1049.45  4911.9 1048.04  4920.5 1046.92  4927.4 1044.77
  4942.9 1043.34  4964.2  1041.8  4985.6 1041.56  4991.4 1040.72  4994.6 1038.51
  4995.6 1038.01  5032.1 1038.51  5035.5 1043.27    5047 1047.47  5068.8 1054.96
  5075.3 1058.57  5113.1 1063.56  5135.3 1067.61  5246.1 1082.35  5412.4 1086.63
#Mann= 6 ,-1 , 0
    4090     .05       0  4099.9     .12       0    4326     .05       0
  4994.6     .05       0  5032.1     .05       0    5047     .12       0
Bank Sta=4994.6,5032.1
XS Rating Curve= 0 ,0
Exp/Cntr=0.3,0.1

Type RM Length L Ch R = 1 ,34726   ,322,322,322
BEGIN DESCRIPTION:
LITTLE LLANO RIVER 63.0
END DESCRIPTION:
XS GIS Cut Line= 3
      2843705.68     10278653.11      2843089.75       10277850.
      2842805.68     10277553.11
#Sta/Elev= 30
  3987.9 1082.44    4016 1082.08  4041.2 1078.94  4115.7 1072.71  4216.6 1067.79
  4358.6 1062.77  4686.8 1062.59  4715.8 1059.73  4757.5 1050.25  4821.8 1050.49
  4936.1 1046.62  4950.6 1041.61  4984.6 1041.73  5031.6 1039.83  5032.5 1039.33
  5069.1 1039.83  5071.4 1047.76  5085.5 1051.15  5092.6 1051.91  5099.7 1048.56
  5106.6 1051.96  5113.9  1051.3  5120.8 1054.77    5128 1053.15  5163.2 1056.49
  5191.5 1063.32  5263.9  1072.1  5326.1  1081.1  5408.2 1082.91  5410.9 1082.91
#Mann= 8 ,-1 , 0
  3987.9     .05       0  4041.2     .12       0  4216.6     .05       0
  4984.6     .12       0  5031.6     .07       0  5069.1     .12       0
  5263.9     .12       0  5408.2     .05       0
Bank Sta=5031.6,5069.1
XS Rating Curve= 0 ,0
Exp/Cntr=0.3,0.1

Type RM Length L Ch R = 1 ,34404   ,286,286,286
BEGIN DESCRIPTION:
Mapping XS 4596b7bb
END DESCRIPTION:
XS GIS Cut Line= 2
      2843986.33     10278334.44      2843032.38     10277337.12
#Sta/Elev= 30
  3962.4 1064.97  3999.2 1063.62  4048.5 1064.71  4204.2 1063.06  4324.4  1060.6
  4614.6 1060.22  4649.9 1060.57  4670.9 1062.08  4727.6 1059.51  4741.7 1056.51
  4755.9 1051.01  4777.3 1047.23  4840.8 1045.96  4876.3  1046.8  4904.6 1045.13
  4932.9 1040.96  4969.7 1038.99  4982.3 1039.06  4984.6 1037.67  4985.6 1037.17
  5022.1 1037.67  5024.8  1038.9  5038.9 1040.76  5053.1 1047.59    5060 1049.66
  5130.8 1066.59    5138 1069.16  5153.5 1071.92  5187.4 1074.29  5342.5 1077.36
#Mann= 5 ,-1 , 0
  3962.4     .05       0  4969.7     .12       0  4984.6     .07       0
  5022.1     .12       0  5153.5     .05       0
Bank Sta=4984.6,5022.1
XS Rating Curve= 0 ,0
Exp/Cntr=0.3,0.1

Type RM Length L Ch R = 1 ,34118   ,267,267,267
BEGIN DESCRIPTION:
Mapping XS 75f2ed68
END DESCRIPTION:
XS GIS Cut Line= 4
      2844420.36     10278117.41       2843986.3     10277965.49
      2843573.98     10277509.76      2843227.01     10277097.74
#Sta/Elev= 30
  3776.4 1065.93  3940.3 1062.37  4105.9 1060.53  4167.9 1060.45  4173.4 1061.56
  4205.1 1060.05  4394.1 1059.08  4684.5 1059.08  4712.5 1060.47  4769.2 1059.53
  4783.4 1058.11  4797.6 1054.09  4805.1 1049.84  4819.3 1045.32  4832.8  1044.3
    4861 1045.41  4897.4 1044.86  4924.9 1038.87  4967.6 1040.81    4971 1034.82
  4971.9 1034.32  5008.5 1034.82  5011.4 1036.16  5021.8 1040.97  5045.7 1048.52
  5074.3 1053.37  5102.9  1062.6  5123.7 1065.15  5209.5 1067.94  5389.5 1068.03
#Mann= 5 ,-1 , 0
  3776.4     .05       0    4971     .05       0  5008.5     .05       0
  5011.4     .12       0  5021.8     .05       0
Bank Sta=4971,5008.5
XS Rating Curve= 0 ,0
Exp/Cntr=0.3,0.1

Type RM Length L Ch R = 1 ,33851   ,646,646,646
BEGIN DESCRIPTION:
Mapping XS aa4b3080
END DESCRIPTION:
XS GIS Cut Line= 4
      2844593.92     10277856.97        2844008.     10277639.97
      2843660.78     10277205.94      2843444.14     10276967.63
#Sta/Elev= 30
    3911 1069.82  4143.7 1060.94  4224.1 1059.29  4517.3 1058.31  4542.9  1059.4
  4598.9 1058.16  4677.3 1058.85  4805.4 1057.82  4819.8 1056.87  4834.2  1051.4
  4848.6 1048.11  4912.6 1043.73  4933.4 1039.13  4968.7 1038.89    4971 1036.84
  4972.3 1035.68  4973.3 1035.18  5009.8 1035.68  5011.9  1037.5  5047.1 1037.62
  5061.5 1039.18  5082.5 1044.63  5101.9 1048.11  5132.8 1053.33  5175.4 1055.83
  5231.5 1061.08  5238.9 1060.32  5245.7 1061.52    5274 1062.22  5413.7 1062.19
#Mann= 5 ,-1 , 0
    3911     .05       0    4971     .12       0  4972.3     .07       0
  5009.8     .12       0  5101.9     .05       0
Bank Sta=4972.3,5009.8
XS Rating Curve= 0 ,0
Exp/Cntr=0.3,0.1

Type RM Length L Ch R = 1 ,33205   ,573,573,573
BEGIN DESCRIPTION:
LITTLE LLANO RIVER 60.0
END DESCRIPTION:
XS GIS Cut Line= 3
      2844805.65     10277053.11        2844267.       10276946.
       2843705.7     10276803.12
#Sta/Elev= 30
  4450.8 1076.21  4476.3 1072.06  4481.4 1072.39  4511.9 1069.19  4694.7 1057.05
    4777 1053.49  4792.1  1051.5  4834.2 1049.85  4839.3 1048.38  4868.8 1044.58
  4899.4 1038.34  4919.8 1036.22  4970.8 1036.66  4998.1 1034.94  5003.1 1033.83
  5004.1 1033.33  5040.9 1033.83  5042.6 1037.12  5063.3 1036.51  5094.2 1038.31
  5135.5 1038.58  5157.4 1042.74    5249 1044.37  5269.6 1046.84  5280.2 1049.23
  5300.6 1050.16  5310.7 1049.66  5351.7 1052.85  5474.4 1055.63  5579.2 1060.37
#Mann= 5 ,-1 , 0
  4450.8     .05       0  4694.7     .12       0  4792.1     .05       0
  5003.1     .05       0  5040.9     .05       0
Bank Sta=5003.1,5040.9
XS Rating Curve= 0 ,0
Exp/Cntr=0.3,0.1

Type RM Length L Ch R = 1 ,32632   ,499,499,499
BEGIN DESCRIPTION:
LITTLE LLANO RIVER 59.0
END DESCRIPTION:
XS GIS Cut Line= 3
      2844755.67     10276253.12      2844412.75       10276465.
      2843755.71     10276603.11
#Sta/Elev= 30
  4596.9 1092.66  4641.2 1091.15  4677.9 1088.14  4699.2 1084.69  4720.4 1083.26
  4757.1 1078.06  4778.4  1076.5  4789.6 1074.71  4808.5 1072.19    4815 1070.16
  4872.9 1063.53  4888.3 1059.74  4894.2 1060.08  4905.5  1052.8    4925  1044.5
  4930.9 1044.43  4946.2 1037.85  4961.3 1035.32  4967.5 1032.99  4969.9 1029.82
  4970.9 1029.32  5007.7 1029.82  5013.7 1033.96  5027.7 1033.66  5068.7 1038.03
  5099.2 1037.47  5140.1 1040.45    5208 1051.33  5538.6 1053.53  5671.4 1058.04
#Mann= 5 ,-1 , 0
  4596.9     .05       0  4789.6     .12       0  4905.5     .05       0
  4969.9     .03       0  5007.7     .05       0
Bank Sta=4969.9,5007.7
XS Rating Curve= 0 ,0
Exp/Cntr=0.3,0.1

Type RM Length L Ch R = 1 ,32133   ,592,592,592
BEGIN DESCRIPTION:
LITTLE LLANO RIVER 58.0
END DESCRIPTION:
XS GIS Cut Line= 3
      2844555.68     10275853.11      2844155.75       10276038.
       2843755.7     10276403.09
#Sta/Elev= 30
  4559.4 1082.05  4596.5 1078.67  4658.5 1070.32  4665.3 1068.75  4716.7 1063.45
  4734.1 1059.82  4739.7 1059.85  4757.1 1055.99  4762.6 1056.24  4768.7 1053.86
  4808.4 1046.14  4824.5 1044.59  4905.7 1038.14  4934.1 1033.76    4980 1032.23
  4989.1 1031.18    4992 1028.96    4993 1028.46  5029.8 1028.96  5031.9 1030.55
  5046.1 1033.79  5074.4 1035.67  5088.6 1038.94  5102.8 1039.74  5109.6 1040.99
  5131.2 1047.68  5145.4 1050.11  5230.2 1051.77  5379.1 1051.71  5541.6 1056.05
#Mann= 4 ,-1 , 0
  4559.4     .12       0  4824.5     .05       0    4992     .03       0
  5029.8     .05       0
Bank Sta=4992,5029.8
XS Rating Curve= 0 ,0
Exp/Cntr=0.3,0.1

Type RM Length L Ch R = 1 ,31541   ,403,403,403
BEGIN DESCRIPTION:
LITTLE LLANO RIVER 57.0
END DESCRIPTION:
XS GIS Cut Line= 3
       2844555.7     10275703.12       2843895.5       10275506.
      2843105.65     10276153.14
#Sta/Elev= 30
    4311 1078.17  4379.1 1071.35  4465.3 1059.88  4519.7 1055.32  4679.8  1046.8
  4712.9 1042.99  4817.5 1036.62  4864.1 1036.89    4889  1035.4  4905.9 1031.66
  4940.9  1030.8  4955.3 1028.51  4978.9 1030.17  4993.6 1029.94  4993.7 1028.39
  4994.7 1027.89  5031.6 1028.39  5033.5 1030.73  5054.3 1030.73  5090.3 1035.81
  5140.4 1035.33  5161.2 1036.92  5208.7 1045.58  5239.5 1048.75  5352.8 1049.93
    5430 1050.39  5607.5 1050.54  5723.2 1052.68  5871.8 1058.38  6021.1 1069.91
#Mann= 9 ,-1 , 0
    4311     .05       0  4379.1     .12       0  4940.9     .05       0
  4993.7     .05       0  5031.6     .05       0  5208.7     .12       0
  5352.8     .05       0    5430     .12       0  5607.5     .05       0
Bank Sta=4993.7,5031.6
XS Rating Curve= 0 ,0
Exp/Cntr=0.3,0.1

Type RM Length L Ch R = 1 ,31138   ,513,513,513
BEGIN DESCRIPTION:
Mapping XS e264f74b
END DESCRIPTION:
XS GIS Cut Line= 2
      2844550.49     10275159.83      2842935.89     10275159.83
#Sta/Elev= 30
  4148.5 1065.65  4343.3 1056.53  4483.3 1051.28  4543.3 1048.16  4623.3 1046.57
  4645.6 1045.04  4703.3 1038.92  4803.3 1034.96  4843.2 1034.65  4893.3 1034.98
  4923.3 1030.79  4941.9 1028.97  4973.3 1029.59  4983.3  1028.7  4994.4 1026.58
  4995.4 1026.08  5031.3 1026.08  5032.3 1026.58  5033.3 1028.05  5043.3 1026.64
  5053.3 1026.84  5063.3 1030.64  5073.3 1035.83  5093.3 1042.85  5133.3 1047.36
  5183.3 1048.09  5253.3  1047.2  5323.3 1047.77  5523.3 1046.92  5763.1 1048.29
#Mann= 6 ,-1 , 0
  4148.5     .12       0  4645.6     .05       0  4843.2     .12       0
  4941.9     .05       0  4994.4     .05       0  5032.3     .05       0
Bank Sta=4994.4,5032.3
XS Rating Curve= 0 ,0
Exp/Cntr=0.3,0.1

Type RM Length L Ch R = 1 ,30625   ,450,450,450
BEGIN DESCRIPTION:
LITTLE LLANO RIVER 55.0
END DESCRIPTION:
XS GIS Cut Line= 3
       2844255.7     10274603.11       2843450.5       10274714.
      2842705.68     10274553.11
#Sta/Elev= 30
  4187.2 1056.81  4516.2 1038.25  4568.4 1037.23  4836.6 1031.18  4975.8 1025.74
  4976.8 1025.24  5013.7 1025.74  5024.1 1033.61  5029.2 1029.55  5045.8 1038.97
  5073.3 1045.35  5137.9 1045.92  5158.4 1041.66  5199.3 1044.21  5209.5 1036.75
    5216 1040.53  5221.1 1038.39    5230 1042.06  5260.1 1046.28    5378 1041.59
  5393.7 1037.83  5414.2 1043.07  5434.6 1043.05  5452.1 1038.17    5463 1039.46
  5470.8 1042.07  5485.8 1045.04  5557.7 1048.85  5710.8 1055.43    5762 1067.59
#Mann= 9 ,-1 , 0
  4187.2     .12       0  4568.4     .05       0  4836.6     .12       0
  4975.8     .05       0  5013.7     .12       0    5378     .12       0
    5463     .05       0  5470.8     .12       0  5557.7     .05       0
Bank Sta=4975.8,5013.7
XS Rating Curve= 0 ,0
Exp/Cntr=0.3,0.1

Type RM Length L Ch R = 1 ,30175   ,1199,1199,1199
BEGIN DESCRIPTION:
LITTLE LLANO RIVER 54.0
END DESCRIPTION:
XS GIS Cut Line= 3
      2844405.65      10274503.1       2843282.5       10274297.
      2842655.72     10274403.11
#Sta/Elev= 30
  3858.1 1062.08  3929.2 1060.61  4288.8 1041.63  4494.4 1032.03  4630.8    1034
  4640.9 1033.51  4658.8 1026.82  4691.8 1026.82  4732.4  1030.8  4762.9 1027.93
  4905.3 1027.78  4966.3 1025.64  4967.6 1022.58  4968.6 1022.08  5005.5 1022.58
  5009.3 1040.17  5017.1 1043.83  5069.7 1043.22  5088.1  1037.7  5098.2  1031.1
  5108.3 1030.59    5125 1040.53  5130.1 1040.46  5138.8 1045.09  5190.5 1040.73
  5219.9 1043.96  5385.4 1050.46    5514 1056.02  5587.3 1064.23  5635.7 1072.15
#Mann= 6 ,-1 , 0
  3858.1     .12       0  4288.8     .05       0  4967.6     .05       0
  5005.5     .05       0  5385.4     .12       0  5587.3     .05       0
Bank Sta=4967.6,5005.5
XS Rating Curve= 0 ,0
Exp/Cntr=0.3,0.1

Type RM Length L Ch R = 1 ,28976   ,703,703,703
BEGIN DESCRIPTION:
Mapping XS fd9d6d5d
END DESCRIPTION:
XS GIS Cut Line= 3
      2844268.84     10274258.86      2843984.25     10273330.56
      2843531.38     10272857.41
#Sta/Elev= 30
  4149.1 1050.33  4315.3 1044.87  4427.1 1043.36  4620.5 1042.38    4762 1044.05
  4814.1 1039.48    4835 1031.91  4866.4 1024.85  4918.7 1022.46  4963.7 1023.84
  4972.9 1023.53  5003.9 1019.58  5004.9 1019.08  5042.6 1019.58  5044.2 1023.64
  5067.1 1022.93    5086 1026.76  5294.1 1042.72  5336.6 1044.18  5343.5 1046.12
  5350.8 1045.43  5379.1 1047.82  5421.2 1053.89  5499.2 1058.59  5555.8 1057.91
    5591 1054.78  5612.4  1054.9    5676 1050.75  5725.6 1049.43    5775 1050.47
#Mann= 5 ,-1 , 0
  4149.1     .05       0  4963.7      .1       0  4972.9     .12       0
  5003.9     .07       0  5042.6     .12       0
Bank Sta=5003.9,5042.6
XS Rating Curve= 0 ,0
Exp/Cntr=0.3,0.1

Type RM Length L Ch R = 1 ,28273   ,595,595,595
BEGIN DESCRIPTION:
LITTLE LLANO RIVER 50.0
END DESCRIPTION:
XS GIS Cut Line= 3
      2844455.69     10274453.09      2844563.75       10273068.
       2844355.7     10272703.15
#Sta/Elev= 30
  3610.7 1060.87  3693.2 1057.73  3941.7 1048.09  4252.6 1041.49  4463.3 1039.89
  4533.5 1042.25  4553.5 1040.75  4623.7 1039.72  4724.1 1040.57  4764.2 1035.11
  4774.2 1030.88  4774.9 1018.59  4775.9 1018.09  4813.6 1018.59  4830.7 1020.42
    4903 1023.12  4984.8 1021.61  4994.9 1018.85  4999.9 1020.36    5052  1020.3
  5074.7 1023.19  5089.1 1022.84  5169.4 1027.22  5209.5  1031.5  5229.2 1033.45
  5258.9 1038.61  5309.8 1039.41  5374.7 1044.69  5411.5 1046.04    5420 1046.72
#Mann= 9 ,-1 , 0
  3610.7     .12       0  3693.2     .05       0  4774.9     .07       0
  4813.6     .05       0    4903     .12       0  5089.1     .05       0
  5169.4     .12       0  5209.5     .05       0  5411.5     .12       0
Bank Sta=4774.9,4813.6
XS Rating Curve= 0 ,0
Exp/Cntr=0.3,0.1

Type RM Length L Ch R = 1 ,27678   ,539,539,539
BEGIN DESCRIPTION:
LITTLE LLANO RIVER 49.0
END DESCRIPTION:
XS GIS Cut Line= 3
      2845005.68     10274353.11        2845082.       10272812.
      2844605.69     10272503.11
#Sta/Elev= 30
    3457 1062.06  3637.2 1053.57  3716.2 1047.81  3847.5 1043.12    4288 1037.51
  4598.4 1037.28  4778.6 1039.29  4798.6 1037.85  4808.7 1033.74  4828.7  1020.9
  4838.7 1017.36  4878.7 1016.84  4888.8 1017.16  4898.8 1019.83  4928.8 1021.41
    4973 1021.22  4978.9 1019.97    4985 1016.16    4986 1015.66  5023.7 1016.16
  5025.5 1018.48  5031.4 1019.14  5061.7 1017.88  5149.4 1022.45  5185.6 1020.75
  5273.7 1034.11  5333.5 1034.92  5388.2  1036.5  5502.7 1041.07  5567.7    1045
#Mann= 9 ,-1 , 0
    3457     .12       0  3716.2     .05       0    4973     .12       0
    4985     .07       0  5023.7     .12       0  5273.7     .05       0
  5333.5     .12       0  5388.2     .05       0  5502.7     .12       0
Bank Sta=4985,5023.7
XS Rating Curve= 0 ,0
Exp/Cntr=0.3,0.1

Type RM Length L Ch R = 1 ,27139   ,524,524,524
BEGIN DESCRIPTION:
LITTLE LLANO RIVER 48.0
END DESCRIPTION:
XS GIS Cut Line= 3
      2846647.18     10273335.65      2845281.91     10272387.21
      2844595.07     10272359.08
#Sta/Elev= 30
  3642.6 1053.96  3690.5 1053.32  3807.6 1050.96  3908.5 1049.04  4249.4 1043.48
  4687.7  1040.9  4747.7 1038.43  4940.4 1035.01  4953.1 1033.24  4959.5 1025.36
    4968 1018.84  4982.8 1015.33  4984.3 1011.93  4985.3 1011.43  5023.1 1011.93
  5024.7  1016.2  5060.5 1017.47    5105 1014.84  5146.9 1016.92  5167.9 1015.39
  5190.8 1018.26  5218.5 1015.82    5284 1019.89  5331.2 1026.49  5361.7  1027.9
    5392 1029.16  5543.1 1034.17  5820.9 1038.02  5919.6 1042.97  5992.4 1046.02
#Mann= 13 ,-1 , 0
  3642.6     .12       0  3690.5     .05       0  3807.6     .12       0
  3908.5     .05       0  4747.7     .12       0  4940.4     .05       0
  4984.3     .05       0  5023.1     .05       0  5361.7     .12       0
    5392     .05       0  5543.1     .12       0  5820.9     .05       0
  5919.6     .12       0
Bank Sta=4984.3,5023.1
XS Rating Curve= 0 ,0
Exp/Cntr=0.3,0.1

Type RM Length L Ch R = 1 ,26615   ,256,256,256
BEGIN DESCRIPTION:
LITTLE LLANO RIVER 47.0
END DESCRIPTION:
XS GIS Cut Line= 3
      2846205.72     10272253.12      2845812.25       10272119.
      2844655.71     10272303.11
#Sta/Elev= 30
  4584.3 1039.02  4756.7 1032.32  4882.1 1031.98  4938.3  1033.3  4954.1 1033.29
  4964.7 1029.23  4976.1  1021.1  4984.7 1010.59  4985.7 1010.09  5028.6 1010.59
    5037 1014.61  5055.1 1015.52  5077.5 1014.67  5117.3 1017.38  5158.5 1015.23
  5184.5  1016.6  5308.9 1014.23  5330.7 1014.68  5350.9  1017.8  5371.1 1019.03
  5411.7 1020.03  5443.4 1019.01  5452.2  1019.7  5492.7 1028.57  5562.7 1032.42
    5675 1031.89  5804.9 1034.46    5967 1035.37  6040.3 1037.28  6171.1 1044.11
#Mann= 7 ,-1 , 0
  4584.3     .12       0  4938.3     .05       0  4984.7     .05       0
  5028.6     .05       0  5804.9     .12       0    5967     .05       0
  6040.3     .12       0
Bank Sta=4984.7,5028.6
XS Rating Curve= 0 ,0
Exp/Cntr=0.3,0.1

Type RM Length L Ch R = 1 ,26359   ,560,560,560
BEGIN DESCRIPTION:
LITTLE LLANO RIVER 46.0
END DESCRIPTION:
XS GIS Cut Line= 3
      2846305.71     10271953.11       2845795.5       10271896.
      2844655.73      10272253.1
#Sta/Elev= 30
  4486.6 1037.73  4526.5 1036.82  4607.4 1035.61  4697.9 1030.54  4818.7 1031.09
  4838.8 1029.71  4874.8 1020.44  4892.6 1017.94  4909.3 1011.28  4939.4 1013.75
  4959.6 1012.93  4960.9 1011.18  4961.9 1010.68  5004.8 1011.18  5031.2 1015.32
  5070.9 1013.86    5157 1014.99  5188.4 1012.44    5206 1014.23  5243.6 1013.98
  5303.3 1017.84  5346.2 1018.15  5373.4 1021.86  5411.1 1022.92  5460.9 1029.37
  5534.3  1032.6  5670.5 1031.61  5836.4 1033.51  6010.8 1035.11  6194.4 1044.44
#Mann= 6 ,-1 , 0
  4486.6     .05       0  4526.5     .12       0  4874.8     .05       0
  4960.9     .05       0  5004.8     .05       0  5836.4     .12       0
Bank Sta=4960.9,5004.8
XS Rating Curve= 0 ,0
Exp/Cntr=0.3,0.1

Type RM Length L Ch R = 1 ,25799   ,477,477,477
BEGIN DESCRIPTION:
LITTLE LLANO RIVER 45.0
END DESCRIPTION:
XS GIS Cut Line= 3
      2846355.72     10271703.13        2845883.       10271399.
      2844605.72     10272203.09
#Sta/Elev= 30
  4437.9 1037.89  4466.7 1037.35  4518.2 1031.94  4609.5 1029.86  4643.7 1029.35
  4684.6 1029.37  4711.7 1019.77  4720.9 1018.01  4770.9  1019.4  4900.3 1016.75
  4953.7 1012.91  4959.9 1012.57  4965.1 1009.64  4966.1 1009.14    5009 1009.64
  5015.8 1011.75  5103.2 1013.55  5210.1 1014.09  5313.7 1011.59  5350.2 1014.86
  5413.8 1015.79  5429.1 1019.74  5471.5 1021.74  5632.8 1021.82  5769.4 1029.74
  5821.2 1031.14  6009.5 1031.11  6065.6 1032.99  6240.3 1034.47  6509.3 1045.08
#Mann= 8 ,-1 , 0
  4437.9     .05       0  4609.5     .12       0  4643.7     .05       0
  4900.3     .12       0  4953.7     .05       0  4965.1     .05       0
    5009     .05       0  6065.6     .12       0
Bank Sta=4965.1,5009
XS Rating Curve= 0 ,0
Exp/Cntr=0.3,0.1

Type RM Length L Ch R = 1 ,25322   ,1070,1070,1070
BEGIN DESCRIPTION:
Mapping XS 2b00403d
END DESCRIPTION:
XS GIS Cut Line= 4
      2846462.98     10270902.61      2845840.59     10270968.12
      2844743.24     10271279.31        2844221.     10271638.35
#Sta/Elev= 30
    4164 1030.67  4271.9 1030.37    4473 1025.62  4716.5 1029.03  4805.3 1030.56
  4817.4 1023.01  4823.7  1016.3  4836.5 1011.73    4930 1012.05  4947.7 1008.78
  4948.7 1008.28  4991.7 1008.78  4992.4 1010.28  5014.1 1010.79  5081.9 1009.67
  5154.9  1011.4  5179.5 1009.37    5228 1012.36  5252.3 1010.31  5273.1 1012.52
    5325  1013.4  5345.8 1015.75  5413.1 1018.39  5699.2 1017.32  5924.4 1029.41
  6002.6 1029.55  6074.4 1027.16    6370 1031.17  6471.5 1034.26  6564.2 1034.15
#Mann= 5 ,-1 , 0
    4164     .05       0  4716.5     .12       0  4817.4     .05       0
  4947.7     .05       0  4991.7     .05       0
Bank Sta=4947.7,4991.7
XS Rating Curve= 0 ,0
Exp/Cntr=0.3,0.1

Type RM Length L Ch R = 1 ,24252   ,752,752,752
BEGIN DESCRIPTION:
Mapping XS 128ec34e
END DESCRIPTION:
XS GIS Cut Line= 3
      2845644.07     10270591.43      2845136.32     10270345.74
      2843662.24     10270493.15
#Sta/Elev= 30
  4226.9 1028.23    4811 1028.38  4892.1 1024.81  4911.2 1021.14  4932.3 1012.74
  4952.4 1009.16  4954.6 1007.26  4960.5 1002.18  4961.5 1001.68  5004.6 1002.18
  5011.7 1005.34    5063 1004.42  5083.1 1005.63  5103.2 1003.68  5163.5 1005.25
  5193.6 1013.69  5223.8 1017.47    5440 1028.39  5505.2 1032.34  5614.7    1035
  5655.9 1039.64  5686.1 1046.62  5706.1  1046.8  5726.2 1050.01  5774.3 1049.04
  5815.7 1042.59  5866.9 1038.53  5947.3  1035.4    6078 1040.81  6272.4 1042.19
#Mann= 7 ,-1 , 0
  4226.9     .05       0    4811     .12       0  4954.6     .05       0
  4960.5     .05       0  5004.6     .05       0    5440     .12       0
  5774.3     .05       0
Bank Sta=4960.5,5004.6
XS Rating Curve= 0 ,0
Exp/Cntr=0.3,0.1

Type RM Length L Ch R = 1 ,23500   ,811,811,811
BEGIN DESCRIPTION:
Mapping XS 52d4e58d
END DESCRIPTION:
XS GIS Cut Line= 3
        2846119.     10269854.39      2845087.18     10269739.74
      2844153.59     10269313.89
#Sta/Elev= 30
  3779.1 1035.84  3922.4 1040.61  4284.6 1026.57  4440.5 1023.65  4556.7 1024.13
  4596.8 1024.23  4728.4 1020.39  4798.7 1015.29  4829.9 1005.21  4845.8 1007.33
  4868.9 1001.98  4874.4 1005.46    4915 1000.22    4938 1002.76  4972.8 1001.54
  4972.9  996.54  4973.9  996.04  5017.3  996.54  5018.1 1000.67    5041  1001.3
  5081.7  999.97  5156.3 1010.84  5195.7 1019.62  5207.9 1020.51  5225.5 1015.56
    5277 1022.71  5378.8 1025.42  5541.5 1028.61  5765.3 1048.87  5843.4 1048.73
#Mann= 10 ,-1 , 0
  3779.1     .05       0  4440.5     .12       0  4556.7     .05       0
  4596.8     .12       0  4728.4     .05       0  4972.9     .03       0
  5017.3     .05       0    5041     .12       0  5195.7     .05       0
  5378.8     .12       0
Bank Sta=4972.9,5017.3
XS Rating Curve= 0 ,0
Exp/Cntr=0.3,0.1

Type RM Length L Ch R = 1 ,22689   ,884,884,884
BEGIN DESCRIPTION:
Mapping XS c809bec5
END DESCRIPTION:
XS GIS Cut Line= 2
      2845988.03     10269395.82      2844743.22     10268593.24
#Sta/Elev= 30
  4213.9  1029.4  4282.8 1030.07  4391.7 1028.53  4774.8 1019.21  4847.3 1018.68
  4875.5  1019.7  4908.2 1018.24  4918.7 1015.51  4942.2 1003.23  4946.9  993.59
  4947.9  993.09  4991.7  993.59  4999.6  995.41  5013.9  995.58  5026.7  997.74
  5049.6  996.73  5072.2 1000.75  5110.8 1003.51  5131.4 1005.76  5156.7 1009.94
  5208.2 1013.77  5216.1 1015.56  5223.4 1013.51  5301.9 1020.79  5353.4 1020.43
    5432 1022.62  5549.3 1026.72  5571.2 1028.54  5598.3 1028.27    5695 1031.77
#Mann= 7 ,-1 , 0
  4213.9     .05       0  4774.8     .12       0  4908.2     .05       0
  4946.9     .05       0  4991.7     .05       0  5110.8     .12       0
  5131.4     .05       0
Bank Sta=4946.9,4991.7
XS Rating Curve= 0 ,0
Exp/Cntr=0.3,0.1

Type RM Length L Ch R = 1 ,21805   ,1015,1015,1015
BEGIN DESCRIPTION:
Mapping XS 6ec60dc5
END DESCRIPTION:
XS GIS Cut Line= 4
      2847200.01     10268871.69      2846037.13     10268380.33
      2845693.18     10268151.04      2844301.04     10268052.77
#Sta/Elev= 30
  3486.8 1029.34  3610.9 1030.83  3931.1 1025.46  3990.9 1021.68  4025.3 1023.28
  4235.9 1017.08  4446.5 1016.44  4555.4 1011.47  4657.2 1016.13  4751.2 1016.63
  4786.4 1013.66  4835.1 1005.11  4914.3 1002.64  4956.9  991.65  4957.9  991.15
  5001.7  991.65  5043.5  996.27  5073.6   993.7  5109.6 1001.06  5136.7 1012.31
  5151.7 1015.44  5180.1 1013.09  5350.9 1019.79  5641.3 1019.58  6062.3 1026.67
  6203.4 1032.01  6302.2 1034.68  6403.2 1041.18  6433.2 1038.88  6558.2 1042.91
#Mann= 11 ,-1 , 0
  3486.8     .05       0  3931.1     .12       0  4025.3     .05       0
  4235.9     .12       0  4446.5     .05       0  4657.2     .12       0
  4786.4     .05       0  4956.9     .05       0  5001.7     .05       0
  6203.4     .12       0  6302.2     .05       0
Bank Sta=4956.9,5001.7
XS Rating Curve= 0 ,0
Exp/Cntr=0.3,0.1

Type RM Length L Ch R = 1 ,20790   ,586,586,586
BEGIN DESCRIPTION:
LITTLE LLANO RIVER 35.0
END DESCRIPTION:
XS GIS Cut Line= 3
       2846405.7     10267603.13      2846138.25       10267301.
      2844382.89     10267348.49
#Sta/Elev= 30
  4596.5 1031.48  4674.7  1030.4  4795.2 1021.75  4858.7 1013.79  4915.6 1004.65
  4922.3 1001.26  4929.9 1001.61  4936.5  996.04  4943.8  995.97  4949.2  989.74
  4950.2  989.24  4994.1  989.74  5022.6  993.68  5042.6  993.71  5052.6   991.1
  5122.6  991.89  5162.6  993.97  5192.6  998.74  5212.6  998.07  5222.6  999.44
  5252.7 1014.28  5265.3 1014.63  5502.7 1012.98  5532.8 1015.11  5562.8 1011.63
  5635.2 1012.21  5682.8 1014.13    6093 1019.46  6543.1 1031.58    6756  1034.7
#Mann= 3 ,-1 , 0
  4596.5     .12       0  4949.2     .05       0  4994.1     .05       0
Bank Sta=4949.2,4994.1
XS Rating Curve= 0 ,0
Exp/Cntr=0.3,0.1

Type RM Length L Ch R = 1 ,20204   ,568,568,568
BEGIN DESCRIPTION:
LITTLE LLANO RIVER 34.0
END DESCRIPTION:
XS GIS Cut Line= 3
      2846405.69     10266953.12        2846061.       10266722.
      2845805.69     10266403.12
#Sta/Elev= 30
    4585 1014.01  4670.6 1010.42  4765.6 1009.05  4843.3  1001.7  4886.7  998.52
  4895.6  992.95  4901.7  993.62  4910.1  990.37  4922.7  988.73  4973.7  989.12
  4988.3  986.47  4989.3  985.97  5033.2  986.47  5039.8  988.76  5081.2  991.19
    5102  988.74    5110  986.55  5124.4  987.55  5130.8  991.05  5138.8  993.17
  5145.2 1000.09  5159.6 1002.54    5166 1005.45  5194.8 1009.44  5246.6 1012.75
  5284.1 1013.75  5351.7 1016.09  5366.1 1017.05  5386.9  1020.8  5408.5 1021.61
#Mann= 7 ,-1 , 0
    4585     .12       0  4843.3     .05       0  4988.3     .05       0
  5033.2     .05       0  5039.8     .12       0  5246.6     .05       0
  5284.1     .12       0
Bank Sta=4988.3,5033.2
XS Rating Curve= 0 ,0
Exp/Cntr=0.3,0.1

Type RM Length L Ch R = 1 ,19636   ,348,348,348
BEGIN DESCRIPTION:
LITTLE LLANO RIVER 33.0
END DESCRIPTION:
XS GIS Cut Line= 3
      2846705.73     10266253.12       2846197.5       10266177.
      2845805.72     10266053.12
#Sta/Elev= 30
  4486.1 1009.74  4520.7 1008.78  4589.9 1005.12    4654 1004.55  4678.3  1005.4
  4698.5 1002.88  4718.1  999.23  4723.1 1000.05  4728.8  998.02  4759.2  993.32
  4809.7  990.71  4850.2   987.3  4856.3  989.06  4910.8  988.91  4920.4   989.8
  4971.5  985.97  4975.8  984.48  4976.8  983.98  5020.9  984.48  5022.9  986.08
  5043.9  984.82  5054.3  989.13  5061.1  996.56  5075.3 1002.25    5131 1009.22
  5169.7 1012.41  5211.7 1014.64  5227.9 1017.34  5253.6 1020.11  5410.9  1025.4
#Mann= 3 ,-1 , 0
  4486.1     .05       0  4975.8     .07       0  5020.9     .12       0
Bank Sta=4975.8,5020.9
XS Rating Curve= 0 ,0
Exp/Cntr=0.3,0.1

Type RM Length L Ch R = 1 ,19288   ,320,320,320
BEGIN DESCRIPTION:
LITTLE LLANO RIVER 32.0
END DESCRIPTION:
XS GIS Cut Line= 3
      2846755.72     10266153.14       2846315.5       10265850.
      2845905.73     10265903.11
#Sta/Elev= 30
  4465.5 1009.01  4487.9 1009.15  4529.8 1006.32  4559.6 1006.26  4631.3 1003.41
  4774.6 1002.07  4810.5  999.98  4817.7  997.96  4825.4  991.91  4840.3  987.18
  4854.1  986.05  4861.2  987.82  4890.5  987.98  4910.8  989.24  4975.5  987.22
  4987.3  983.48  4988.3  982.98  5032.4  983.48  5040.1  985.44  5059.2  987.81
  5064.2  986.89  5080.5  995.78  5100.7 1001.75  5120.8 1005.79  5184.3 1009.12
  5222.7 1012.63  5284.5 1014.57  5291.9  1013.9  5312.4 1015.95  5413.2  1020.2
#Mann= 6 ,-1 , 0
  4465.5     .05       0  4910.8     .12       0  4987.3     .07       0
  5032.4     .12       0  5184.3     .05       0  5284.5     .12       0
Bank Sta=4987.3,5032.4
XS Rating Curve= 0 ,0
Exp/Cntr=0.3,0.1

Type RM Length L Ch R = 1 ,18968   ,793,793,793
BEGIN DESCRIPTION:
LITTLE LLANO RIVER 31.0
END DESCRIPTION:
XS GIS Cut Line= 3
      2846955.68     10265703.11       2846433.5       10265552.
      2846055.68     10265403.11
#Sta/Elev= 30
  4456.4 1009.59  4550.8 1006.46  4591.7 1002.69  4664.6  999.48  4768.7  997.79
  4820.8  998.12  4888.8  996.36  4907.7  994.22  4924.9  987.78  4935.3   986.2
  4946.5  985.95  4956.1  984.43  4966.5  985.38    5000  984.05  5004.9  982.71
  5005.9  982.21  5054.8  982.71    5061  987.28  5066.3  988.04  5096.1 1000.17
  5120.5 1006.11  5126.6 1008.57  5144.9 1011.43  5198.9 1016.55  5253.2 1017.66
  5266.4 1016.87  5282.9 1017.84  5303.3 1017.33  5330.9 1015.96  5406.1  1018.4
#Mann= 6 ,-1 , 0
  4456.4     .05       0  4888.8     .12       0  5004.9     .07       0
  5054.8     .12       0  5198.9     .05       0  5303.3     .12       0
Bank Sta=5004.9,5054.8
XS Rating Curve= 0 ,0
Exp/Cntr=0.3,0.1

Type RM Length L Ch R = 1 ,18175   ,595,595,595
BEGIN DESCRIPTION:
LITTLE LLANO RIVER 29.0
END DESCRIPTION:
XS GIS Cut Line= 3
      2847155.71     10265203.13      2846791.25       10264854.
      2846405.72     10264703.13
#Sta/Elev= 30
  4495.3 1007.84  4594.2 1004.34  4700.5  995.83  4735.8  994.49  4764.1  988.78
  4870.1  991.22  4897.9  990.06  4905.6  989.22  4919.7  984.81  4933.9  983.08
  4976.3  983.45  5013.2  981.32  5014.2  980.82  5063.1  981.32    5068  991.05
  5073.4  993.96  5091.9  993.54  5113.4  999.05  5122.3  999.65  5127.7 1001.93
  5134.8  998.77  5152.2  998.26  5176.6 1000.91  5220.7  1001.3  5242.2 1003.72
  5294.2 1003.48  5338.9  1005.1  5374.7 1009.26  5381.8 1011.41    5414 1014.64
#Mann= 5 ,-1 , 0
  4495.3     .05       0  4897.9     .12       0  5013.2     .07       0
  5063.1     .12       0  5294.2     .05       0
Bank Sta=5013.2,5063.1
XS Rating Curve= 0 ,0
Exp/Cntr=0.3,0.1

Type RM Length L Ch R = 1 ,17580   ,598,598,598
BEGIN DESCRIPTION:
LITTLE LLANO RIVER 28.0
END DESCRIPTION:
XS GIS Cut Line= 3
      2847605.68     10264753.11      2847096.75       10264347.
      2846705.66     10264253.11
#Sta/Elev= 30
  4348.9 1007.61    4449 1003.92  4469.8 1004.22  4484.2 1002.91  4562.7 1002.15
  4690.8  996.39  4719.6  995.65  4740.4  996.72  4754.8  994.28  4779.3  992.98
  4833.3  990.57    4851  988.73  4897.3  983.37  4918.2  982.41  4953.4  982.39
  4961.4  981.34  5003.1  980.91  5012.5  979.92  5013.5  979.42  5062.7  979.92
  5062.8  982.82  5079.6  984.95  5140.4  988.62  5196.5  992.15  5217.1  992.25
  5247.5  996.48  5311.1 1000.08    5361    1004  5378.6 1006.88  5402.2 1008.54
#Mann= 8 ,-1 , 0
  4348.9     .12       0  4779.3      .1       0    4851     .12       0
  4918.2     .05       0  5012.5     .05       0  5062.7     .05       0
  5140.4     .12       0  5311.1     .05       0
Bank Sta=5012.5,5062.7
XS Rating Curve= 0 ,0
Exp/Cntr=0.3,0.1

Type RM Length L Ch R = 1 ,16982   ,593,593,593
BEGIN DESCRIPTION:
LITTLE LLANO RIVER 27.0
END DESCRIPTION:
XS GIS Cut Line= 3
      2848055.67     10263953.11      2847273.75       10263784.
      2846505.65     10263853.11
#Sta/Elev= 30
    4200  1016.1  4206.8 1015.45  4219.5 1013.58  4224.6 1014.12  4268.7 1010.52
  4411.3  1003.2  4504.6  999.99  4563.6  999.62  4647.2  995.43  4763.8  994.31
    4839   994.2  4875.2  995.71  4888.3  987.48  4895.7  981.39  4901.3  978.96
  4902.3  978.46  4951.6  978.96  5068.3  980.61  5098.5  981.85  5148.7  986.66
  5218.9  985.94  5271.6   991.9  5289.2  994.87  5362.5  997.81  5382.6  999.07
    5462  998.21  5590.8  1000.7  5630.4 1003.09  5760.7 1010.61  5771.2 1010.85
#Mann= 11 ,-1 , 0
    4200     .05       0  4206.8     .12       0  4563.6     .05       0
  4763.8     .12       0  4901.3     .07       0  4951.6     .12       0
  5362.5     .12       0    5462     .05       0  5590.8     .12       0
  5630.4     .05       0  5760.7     .12       0
Bank Sta=4901.3,4951.6
XS Rating Curve= 0 ,0
Exp/Cntr=0.3,0.1

Type RM Length L Ch R = 1 ,16389   ,1073,1073,1073
BEGIN DESCRIPTION:
LITTLE LLANO RIVER 26.0
END DESCRIPTION:
XS GIS Cut Line= 3
      2847955.72     10263403.13        2847371.       10263204.
      2846655.66     10262453.09
#Sta/Elev= 30
  4382.3  1005.5  4498.5  997.68  4549.5  998.14    4769  989.58  4935.5  979.06
  4973.5  976.99  4979.1  976.35  4980.1  975.85  5029.4  976.35    5051  977.69
  5130.7  980.86    5167  983.67  5188.3  988.05  5322.6  988.71    5344  986.19
  5350.9  987.79  5358.2  984.04  5365.1  986.08  5372.3  981.71  5379.2  983.65
  5386.5  979.78  5443.1  976.85  5506.6  977.47  5534.9  983.34  5584.3  983.93
  5612.6  991.37  5711.7  992.82  5775.2  998.99    5866 1003.33  6037.1 1012.43
#Mann= 8 ,-1 , 0
  4382.3     .05       0  4935.5     .12       0  4973.5     .05       0
  4979.1     .05       0  5029.4     .05       0    5051     .12       0
  5130.7     .05       0    5866     .12       0
Bank Sta=4979.1,5029.4
XS Rating Curve= 0 ,0
Exp/Cntr=0.3,0.1

Type RM Length L Ch R = 1 ,15316   ,668,668,668
BEGIN DESCRIPTION:
LITTLE LLANO RIVER 24.0
END DESCRIPTION:
XS GIS Cut Line= 3
      2848055.66      10262453.1      2847478.75       10262158.
      2846655.67     10262403.12
#Sta/Elev= 30
    4352 1003.37  4449.1  996.42  4604.6  992.58  4643.4  989.54    4649  990.24
  4732.3  987.96  4752.8  986.17  4782.3  980.85  4812.5  977.83  4821.1  975.15
  4826.7  976.48    4835  973.15  4901.8  973.61  4924.8  975.45    4960  976.18
  4969.7  972.26  4971.1  971.36  5026.5  971.36  5027.8  972.26  5032.4  975.18
  5055.4  973.83  5109.1  978.94  5149.3  979.34    5191  982.38  5208.6  988.68
  5337.1  989.71  5522.7   995.2  5532.8  995.29  5698.8 1002.56  5858.8 1011.82
#Mann= 8 ,-1 , 0
    4352     .05       0  4752.8     .12       0  4901.8     .05       0
  4969.7     .05       0  5027.8     .05       0  5522.7     .12       0
  5532.8     .05       0  5698.8     .12       0
Bank Sta=4969.7,5027.8
XS Rating Curve= 0 ,0
Exp/Cntr=0.3,0.1

Type RM Length L Ch R = 1 ,14648   ,1184,1184,1184
BEGIN DESCRIPTION:
Mapping XS be20f9de
END DESCRIPTION:
XS GIS Cut Line= 3
      2848461.17     10262288.93      2847836.14     10261643.06
      2847004.49     10261227.23
#Sta/Elev= 30
  4089.1 1002.95  4344.7  997.26  4535.6  997.19  4678.7  992.37  4770.5  991.24
  4832.7  989.39    4861  985.81  4875.1  985.48  4878.8  986.81  4882.1  987.99
  4889.3   986.9  4896.2  983.64  4924.4  983.11  4952.8  973.22  4955.5  969.39
  4956.9  968.49  5013.7  969.39  5018.8  971.25  5077.8  973.29  5167.3  974.13
    5248  971.28  5268.4  973.98  5287.2  980.31  5309.5  985.65  5376.6  989.41
  5471.6   991.9  5583.4 1000.28  5668.3 1002.94  5762.3  1009.2  5917.7 1013.65
#Mann= 9 ,-1 , 0
  4089.1     .05       0  4678.7     .12       0  4770.5     .05       0
  4878.8     .12       0  4924.4     .05       0  4955.5     .05       0
  5013.7     .05       0  5268.4     .12       0  5668.3     .05       0
Bank Sta=4955.5,5013.7
XS Rating Curve= 0 ,0
Exp/Cntr=0.3,0.1

Type RM Length L Ch R = 1 ,13464   ,383,383,383
BEGIN DESCRIPTION:
Mapping XS 207eea47
END DESCRIPTION:
XS GIS Cut Line= 3
      2848898.63     10262038.85      2848502.81     10260809.73
       2848190.5     10260372.49
#Sta/Elev= 30
  3792.5 1002.68  3903.6  998.36  4124.2  994.78  4179.6  991.73  4345.2  988.64
    4372  984.06  4397.4  984.26  4428.9  987.86  4500.3  985.59  4601.8  986.76
  4817.6  984.97  4863.6  979.78  4870.1  975.61  4890.4  971.15  4933.1  970.59
  4985.3  967.11  5009.1  965.79  5010.5  964.89  5067.4  965.79  5069.7  970.84
  5091.2  973.83  5128.8  977.37  5243.9  982.16  5273.4  985.36  5323.8  986.08
  5374.2  991.25  5436.8   995.3  5466.3   999.7  5522.9 1003.24  5621.1 1004.72
#Mann= 5 ,-1 , 0
  3792.5     .05       0  4985.3     .12       0  5009.1     .07       0
  5067.4     .12       0  5091.2     .05       0
Bank Sta=5009.1,5067.4
XS Rating Curve= 0 ,0
Exp/Cntr=0.3,0.1

Type RM Length L Ch R = 1 ,13081   ,446,446,446
BEGIN DESCRIPTION:
Mapping XS e59192b8
END DESCRIPTION:
XS GIS Cut Line= 3
      2849273.64     10261372.23      2848773.64     10260559.73
      2848190.48     10260184.84
#Sta/Elev= 30
  4203.4 1000.36  4345.9  999.29  4419.3  994.07  4471.4   995.3  4556.5  987.13
  4629.9  986.51  4703.3  979.43  4724.5   975.3    4740  975.61  4767.1  970.92
  4789.5   974.2  4819.2  969.68  4877.2  970.25  4892.6  968.02  4913.9  970.31
  4967.5  967.92  5006.9   965.4  5008.3   964.5  5065.2   965.4  5066.5  973.04
  5094.7  975.15  5190.7  977.38  5402.7  987.21  5493.5  986.92  5508.7  989.92
  5535.8  989.13  5581.7  993.53  5623.7  996.94  5821.4 1003.55  5850.7 1002.31
#Mann= 7 ,-1 , 0
  4203.4     .05       0  4967.5     .12       0  5006.9     .07       0
  5065.2     .12       0  5402.7     .05       0  5581.7     .12       0
  5821.4     .05       0
Bank Sta=5006.9,5065.2
XS Rating Curve= 0 ,0
Exp/Cntr=0.3,0.1

Type RM Length L Ch R = 1 ,12635   ,728,728,728
BEGIN DESCRIPTION:
LITTLE LLANO RIVER 19.0
END DESCRIPTION:
XS GIS Cut Line= 3
      2849255.68     10260853.11      2849155.75       10260368.
      2848405.65      10260103.1
#Sta/Elev= 30
  4504.7  991.16  4580.2  988.65  4623.4  985.89  4719.1  980.64  4739.5  977.79
  4770.2  978.47  4776.6  977.26  4790.6   975.4    4811  970.43  4825.8  969.37
  4831.7  967.42  4851.8  965.66  4876.9  967.46  4913.1  967.41  4914.5  965.02
  4915.9  964.12  4971.6  964.12    4973  965.02  4977.5  966.55  4984.6  966.73
  5028.1  965.64  5093.5  966.36  5127.3  967.05  5146.5  971.47  5177.5  975.45
  5337.6   981.6  5506.4  987.34  5630.7  992.72  5749.1 1002.94  5795.5    1005
#Mann= 9 ,-1 , 0
  4504.7     .05       0  4623.4     .12       0  4776.6     .05       0
  4825.8     .12       0  4914.5     .07       0    4973     .12       0
  5093.5     .05       0  5337.6     .12       0  5506.4     .05       0
Bank Sta=4914.5,4973
XS Rating Curve= 0 ,0
Exp/Cntr=0.3,0.1
