--- LITTLE LLANO RIVER.prj (project) ---

Proj Title=LITTLE LLANO RIVER Base Level Engineering
Current Plan=p01
Default Exp/Contr=0.3,0.1
English Units
Geom File=g01
Flow File=f01
Plan File=p01
BEGIN DESCRIPTION:
LITTLE LLANO RIVER
END DESCRIPTION:

--- LITTLE LLANO RIVER.p01 (plan) ---

Plan Title=Multiple Run
Short Identifier=Multiple
Geom File=g01
Flow File=f01
Subcritical Flow
K Sum by GR= 0
Std Step Tol= 0.01
Critical Tol= 0.01
Num of Std Step Trials= 20
Max Error Tol= 0.3
Flow Tol Ratio= 0.001
Split Flow NTrial= 30
Split Flow Tol= 0.02
Split Flow Ratio= 0.02
Log Output Level= 0
Friction Slope Method= 1
Unsteady Friction Slope Method= 2
Unsteady Bridges Friction Slope Method= 1
Parabolic Critical Depth
Global Vel Dist=  1 , 1 , 1
Global Log Level= 0
CheckData=True
Encroach Param= -1, 0, 0, 0
BEGIN DESCRIPTION:
Multiple Run
END DESCRIPTION:

--- LITTLE LLANO RIVER.f01 (steady flow) ---

Flow Title=Multiple
Number of Profiles=7
Profile Names=10-year,25-year,50-year,1pct_min,100-year,1pct_plu,500-year
River Rch & RM= LITTLE LLANO RIV,Reach-1,65874
     290     653    1101     607    1833    5537    5398
River Rch & RM= LITTLE LLANO RIV,Reach-1,64348
     360     822    1394     774    2337    7057    6961
River Rch & RM= LITTLE LLANO RIV,Reach-1,60954
     377     862    1465     814    2458    7423    7340
River Rch & RM= LITTLE LLANO RIV,Reach-1,56934
     464    1073    1835    1025    3096    9350    9341
River Rch & RM= LITTLE LLANO RIV,Reach-1,55401
     485    1124    1924    1076    3249    9812    9824
River Rch & RM= LITTLE LLANO RIV,Reach-1,51693
     500    1161    1990    1114    3364   10158   10186
River Rch & RM= LITTLE LLANO RIV,Reach-1,45683
     520    1209    2074    1162    3510   10600   10648
River Rch & RM= LITTLE LLANO RIV,Reach-1,42195
     532    1239    2127    1193    3602   10877   10939
River Rch & RM= LITTLE LLANO RIV,Reach-1,36308
     549    1280    2199    1234    3726   11251   11331
River Rch & RM= LITTLE LLANO RIV,Reach-1,35162
     669    1574    2718    1532    4626   13969   14191
River Rch & RM= LITTLE LLANO RIV,Reach-1,28976
     677    1593    2752    1551    4685   14147   14379
River Rch & RM= LITTLE LLANO RIV,Reach-1,27209
     790    1869    3240    1833    5535   16714   17095
River Rch & RM= LITTLE LLANO RIV,Reach-1,22689
     796    1885    3269    1849    5585   16866   17256
River Rch & RM= LITTLE LLANO RIV,Reach-1,18968
     796    1885    3270    1850    5587   16872   17262
River Rch & RM= LITTLE LLANO RIV,Reach-1,18175
     895    2128    3700    2098    6336   19133   19664
River Rch & RM= LITTLE LLANO RIV,Reach-1,15316
    1055    2524    4404    2505    7565   22847   23622
River Rch & RM= LITTLE LLANO RIV,Reach-1,11907
    1103    2642    4614    2627    7933   23957   24808
River Rch & RM= LITTLE LLANO RIV,Reach-1,6358
    1118    2678    4679    2664    8046   24299   25174
Boundary for River Rch & Prof#=LITTLE LLANO RIV,Reach-1,1
Up Type=0
Dn Type=3
Dn Slope=0.005
Boundary for River Rch & Prof#=LITTLE LLANO RIV,Reach-1,2
Up Type=0
Dn Type=3
Dn Slope=0.005
Boundary for River Rch & Prof#=LITTLE LLANO RIV,Reach-1,3
Up Type=0
Dn Type=3
Dn Slope=0.005
Boundary for River Rch & Prof#=LITTLE LLANO RIV,Reach-1,4
Up Type=0
Dn Type=3
Dn Slope=0.005
Boundary for River Rch & Prof#=LITTLE LLANO RIV,Reach-1,5
Up Type=0
Dn Type=3
Dn Slope=0.005
Boundary for River Rch & Prof#=LITTLE LLANO RIV,Reach-1,6
Up Type=0
Dn Type=3
Dn Slope=0.005
Boundary for River Rch & Prof#=LITTLE LLANO RIV,Reach-1,7
Up Type=0
Dn Type=3
Dn Slope=0.005

--- LITTLE LLANO RIVER.g01 (geometry) ---

Geom Title=Existing Conditions

River Reach=LITTLE LLANO RIV,Reach-1
Reach XY= 30
      2832357.50     10303059.00      2832329.50     10301442.00
      2833527.25     10299084.00      2834520.50     10298838.00
      2836119.50     10296602.00      2836878.00     10292399.00
      2837992.75     10290760.00      2836919.75     10289784.00
      2836947.50     10289184.00      2838971.75     10287743.00
      2838652.25     10286791.00      2839815.50     10284055.00
      2839655.75     10282774.00      2842301.75     10281128.00
      2842862.00     10280157.00      2842877.75     10278231.00
      2844442.00     10276811.00      2843298.25     10274097.00
      2845859.50     10272007.00      2844818.25     10269910.00
      2846051.50     10267793.00      2847522.50     10261924.00
      2849322.50     10260006.00      2848768.50     10258418.00
      2849002.75     10257003.00      2851319.00     10255635.00
      2851090.75     10254542.00      2849509.50     10254355.00
      2850715.75     10252949.00      2850685.50     10251651.00

Type RM Length L Ch R = 1,65874,405,405,405
BEGIN DESCRIPTION:
LITTLE LLANO RIVER 125.0
END DESCRIPTION:
XS GIS Cut Line= 3
      2832555.71     10302803.13      2832329.50     10302640.00
      2832005.66     10302453.10
#Sta/Elev= 30
  4721.1 1230.46  4801.1 1229.70  4829.1 1229.27  4843.8 1225.36  4864.7 1221.88
  4870.9 1222.94  4879.4 1222.64  4885.6 1225.04  4893.7 1223.90  4900.3 1221.57
  4906.4 1221.86  4914.3 1219.56  4965.3 1213.43  4986.2 1213.15  5013.8 1210.95
  5014.3 1210.45  5031.8 1210.95  5038.5 1213.03  5044.3 1213.00  5060.1 1219.28
  5065.9 1218.24  5073.7 1221.87  5081.6 1223.74  5205.1 1227.70  5220.9 1229.29
  5235.3 1228.30  5242.5 1230.01  5285.6 1232.45  5338.7 1237.86  5373.9 1242.57
#Mann=5,-1,0
  4721.1    0.05       0  4801.1    0.12       0  4914.3    0.05       0
  5013.8    0.05       0  5031.8    0.05       0
Bank Sta=5013.8,5031.8
Exp/Cntr=0.3,0.1

Type RM Length L Ch R = 1,65469,404,404,404
BEGIN DESCRIPTION:
LITTLE LLANO RIVER 124.0
END DESCRIPTION:
XS GIS Cut Line= 3
      2832905.64     10302503.09      2832371.00     10302237.00
      2831905.66     10302403.12
#Sta/Elev= 30
  4402.8 1233.68  4405.5 1233.68  4411.2 1230.44  4416.7 1229.17  4433.5 1227.78
  4707.8 1226.07  4804.9 1227.39  4864.6 1226.25  4909.4 1224.06  4931.8 1221.51
  4948.6 1216.61  4954.1 1216.95  4971.0 1212.04  4983.6 1209.98  4984.3 1206.83
  4984.8 1206.33  5002.3 1206.83  5010.8 1207.86  5026.9 1209.57  5080.0 1221.37
  5206.8 1227.32  5228.6 1226.81  5272.8 1231.34  5292.3 1233.87  5305.7 1239.16
  5330.0 1238.13  5360.8 1239.59  5422.4 1245.17  5478.7 1253.35  5494.1 1253.35
#Mann=7,-1,0
  4402.8    0.05       0  4804.9    0.12       0  4984.3    0.07       0
  5002.3    0.12       0  5010.8    0.05       0  5272.8    0.12       0
  5305.7    0.05       0
Bank Sta=4984.3,5002.3
Exp/Cntr=0.3,0.1

Type RM Length L Ch R = 1,65065,717,717,717
BEGIN DESCRIPTION:
LITTLE LLANO RIVER 123.0
END DESCRIPTION:
XS GIS Cut Line= 3
      2832955.70     10302353.13      2832371.00     10301834.00
      2832005.71     10302103.09
#Sta/Elev= 30
  4218.1 1228.73  4282.1 1226.98  4572.3 1224.10  4748.5 1224.79  4834.0 1224.81
  4890.9 1222.41  4919.3 1217.50  4940.2 1212.37  4947.8 1208.08  4953.0 1203.54
  4953.5 1203.04  4971.0 1203.54  5000.0 1205.82  5003.7 1207.45  5018.3 1207.35
  5043.0 1211.71  5048.7 1212.40  5060.0 1213.28  5089.3 1218.96  5110.1 1220.02
  5124.8 1222.97  5175.4 1224.19  5254.3 1223.61  5275.2 1225.51  5304.5 1224.85
  5339.9 1226.17  5346.2 1227.91  5360.8 1228.09  5396.3 1235.70  5453.7 1238.93
#Mann=7,-1,0
  4218.1    0.05       0  4748.5    0.12       0  4953.0    0.05       0
  4971.0    0.12       0  5043.0    0.12       0  5048.7    0.05       0
  5175.4    0.12       0
Bank Sta=4953,4971
Exp/Cntr=0.3,0.1

Type RM Length L Ch R = 1,64348,557,557,557
BEGIN DESCRIPTION:
Mapping XS 3736d8a2
END DESCRIPTION:
XS GIS Cut Line= 3
      2833070.52     10301468.10      2832723.28     10301164.27
      2831573.12     10301099.17
#Sta/Elev= 30
  4249.4 1219.78  4447.7 1218.37  4639.4 1222.22  4788.5 1217.19  4860.7 1217.44
  4908.7 1213.19  4928.7 1213.31  4958.8 1204.04  4978.8 1201.15  4985.4 1196.81
  4985.9 1196.31  5005.2 1196.81  5008.9 1199.91  5057.3 1209.00  5079.0 1215.12
  5099.0 1218.16  5189.2 1224.56  5229.2 1226.04  5269.3 1230.35  5308.0 1231.77
  5352.5 1238.26  5369.4 1238.23  5479.6 1247.04  5569.8 1248.12  5664.1 1251.95
  5704.8 1250.99  5760.1 1242.87  5790.1 1240.45  5861.5 1239.92  5862.8 1239.92
#Mann=8,-1,0
  4249.4    0.05       0  4860.7    0.12       0  4985.4    0.07       0
  5005.2    0.12       0  5057.3    0.05       0  5308.0    0.12       0
  5664.1    0.05       0  5861.5    0.12       0
Bank Sta=4985.4,5005.2
Exp/Cntr=0.3,0.1

Type RM Length L Ch R = 1,63791,489,489,489
BEGIN DESCRIPTION:
LITTLE LLANO RIVER 120.0
END DESCRIPTION:
XS GIS Cut Line= 3
      2833555.71     10301203.13      2832732.25     10300682.00
      2832155.71     10300103.13
#Sta/Elev= 30
  4025.5 1232.96  4026.2 1232.96  4039.1 1233.58  4061.0 1232.35  4112.0 1222.86
  4117.7 1220.75  4127.2 1218.71  4179.0 1215.59  4184.9 1216.88  4257.8 1216.90
  4424.8 1214.92  4901.3 1214.98  4924.9 1213.18  4974.0 1199.92  5000.0 1198.18
  5001.0 1194.80  5001.5 1194.30  5020.8 1194.80  5039.2 1200.92  5046.3 1205.89
  5067.5 1210.54  5109.9 1213.97  5449.3 1231.25  5608.9 1244.56  5703.9 1256.19
  5767.5 1268.02  5802.9 1276.20  5810.0 1276.77  5813.5 1279.64  5817.0 1279.64
#Mann=6,-1,0
  4025.5    0.05       0  4026.2    0.12       0  4117.7    0.05       0
  5001.0    0.03       0  5020.8    0.05       0  5608.9    0.12       0
Bank Sta=5001,5020.8
Exp/Cntr=0.3,0.1

Type RM Length L Ch R = 1,63302,410,410,410
BEGIN DESCRIPTION:
LITTLE LLANO RIVER 119.0
END DESCRIPTION:
XS GIS Cut Line= 3
      2833105.72     10300403.15      2832968.25     10300255.00
      2832355.70     10299753.12
#Sta/Elev= 30
  4797.9 1212.97  4863.5 1211.81  4896.9 1211.86  4932.6 1207.55  4960.9 1201.18
  4967.7 1198.05  4981.9 1194.38  5000.4 1191.55  5000.9 1191.05  5020.3 1191.55
  5024.7 1194.33  5045.5 1198.46  5053.4 1202.63  5059.8 1204.05  5067.7 1207.85
  5117.3 1213.64  5138.1 1214.87  5158.9 1218.26  5173.1 1218.17  5237.1 1223.41
  5301.0 1231.22  5424.2 1243.89  5443.1 1247.77  5500.5 1254.22  5564.4 1266.80
  5613.9 1278.37  5677.8 1296.28  5717.6 1305.42  5778.3 1320.08  5791.9 1322.20
#Mann=7,-1,0
  4797.9    0.05       0  4863.5    0.12       0  5000.4    0.07       0
  5020.3    0.12       0  5173.1    0.05       0  5424.2    0.12       0
  5717.6    0.05       0
Bank Sta=5000.4,5020.3
Exp/Cntr=0.3,0.1

Type RM Length L Ch R = 1,62892,511,511,511
BEGIN DESCRIPTION:
LITTLE LLANO RIVER 118.0
END DESCRIPTION:
XS GIS Cut Line= 3
      2833305.67     10300103.08      2833204.50     10299921.00
      2832655.68     10299453.11
#Sta/Elev= 30
  4791.7 1210.80  4871.6 1212.27  4902.6 1210.74  4924.4 1207.43  4946.1 1198.01
  4957.9 1190.20  4958.4 1189.70  4977.8 1190.20  4995.9 1191.98  5011.6 1191.08
  5054.1 1198.63  5061.8 1201.74  5076.1 1204.90  5141.0 1209.96  5210.0 1215.24
  5252.9 1213.99  5260.6 1216.51  5274.4 1218.66  5316.6 1221.39  5373.8 1226.92
  5394.5 1228.24  5437.4 1235.09  5486.8 1248.38  5572.4 1269.62  5636.1 1287.06
  5642.7 1287.53  5671.2 1295.67  5699.8 1301.05  5717.9 1306.70  5721.2 1306.70
#Mann=6,-1,0
  4791.7    0.05       0  4871.6    0.12       0  4957.9    0.07       0
  4977.8    0.12       0  5141.0    0.05       0  5373.8    0.12       0
Bank Sta=4957.9,4977.8
Exp/Cntr=0.3,0.1

Type RM Length L Ch R = 1,62381,914,914,914
BEGIN DESCRIPTION:
LITTLE LLANO RIVER 117.0
END DESCRIPTION:
XS GIS Cut Line= 3
      2833805.69     10299903.12      2833461.25     10299484.00
      2833055.67     10299253.10
#Sta/Elev= 30
  4457.5 1216.20  4571.6 1214.80  4702.2 1209.54  4791.9 1207.36  4798.3 1208.23
  4862.2 1206.72  4919.6 1207.24  4926.1 1202.02  4933.9 1198.36  4940.4 1191.83
  4958.8 1185.46  4959.3 1184.96  4979.3 1185.46  4983.4 1190.60  5040.9 1192.08
  5087.0 1194.81  5092.7 1197.06  5108.6 1199.70  5154.6 1204.52  5216.7 1209.06
  5248.1 1209.30  5275.7 1212.65  5297.4 1216.72  5334.8 1228.81  5356.4 1233.99
  5376.5 1241.15  5421.3 1255.09  5453.0 1263.12  5458.8 1263.12  5466.7 1265.17
#Mann=6,-1,0
  4457.5    0.05       0  4702.2    0.12       0  4958.8    0.07       0
  4979.3    0.12       0  5154.6    0.05       0  5376.5    0.12       0
Bank Sta=4958.8,4979.3
Exp/Cntr=0.3,0.1

Type RM Length L Ch R = 1,61467,513,513,513
BEGIN DESCRIPTION:
LITTLE LLANO RIVER 115.0
END DESCRIPTION:
XS GIS Cut Line= 3
      2834655.67     10299503.10      2833964.75     10298932.00
      2833155.65     10298153.08
#Sta/Elev= 30
  4103.6 1246.03  4265.7 1232.28  4330.9 1229.24  4373.9 1223.16  4594.1 1205.87
  4650.0 1197.10  4686.6 1186.42  4693.0 1187.51  4707.4 1196.71  4736.0 1199.94
  4799.9 1197.34  4849.4 1185.55  4863.7 1188.13  4898.9 1184.03  5002.8 1183.07
  5044.6 1179.85  5045.1 1179.35  5065.5 1179.85  5111.6 1191.66  5118.8 1190.62
  5125.8 1194.27  5161.3 1193.36  5224.8 1201.77  5536.5 1207.65  5645.1 1207.39
  5804.7 1209.41  5911.1 1218.45  5988.6 1242.77  6038.3 1252.43  6123.1 1279.53
#Mann=7,-1,0
  4103.6    0.12       0  4265.7    0.05       0  5044.6    0.03       0
  5065.5    0.05       0  5536.5    0.12       0  5645.1    0.05       0
  5911.1    0.12       0
Bank Sta=5044.6,5065.5
Exp/Cntr=0.3,0.1

Type RM Length L Ch R = 1,60954,514,514,514
BEGIN DESCRIPTION:
LITTLE LLANO RIVER 114.0
END DESCRIPTION:
XS GIS Cut Line= 3
      2834755.67     10299153.10      2834444.00     10298900.00
      2833755.72     10298503.13
#Sta/Elev= 30
  4598.5 1240.45  4640.9 1236.33  4784.5 1218.80  4826.2 1213.26  4832.7 1211.60
  4875.8 1207.76  4890.1 1204.83  4904.5 1201.07  4939.7 1189.30  4954.1 1182.71
  4964.2 1176.26  4964.7 1175.76  4985.5 1176.26  4989.3 1179.36  5019.6 1179.41
  5062.7 1181.13  5078.5 1182.87  5090.4 1185.98  5100.0 1189.87  5105.8 1193.69
  5113.5 1196.88  5127.4 1198.64  5201.6 1201.77  5325.6 1200.96  5610.0 1202.86
  5668.9 1201.85  5700.4 1203.56  5727.8 1202.90  5743.5 1204.32  5794.5 1204.48
#Mann=5,-1,0
  4598.5    0.05       0  4784.5    0.12       0  4964.2    0.07       0
  4985.5    0.12       0  5201.6    0.05       0
Bank Sta=4964.2,4985.5
Exp/Cntr=0.3,0.1

Type RM Length L Ch R = 1,60440,480,480,480
BEGIN DESCRIPTION:
Mapping XS 714aad33
END DESCRIPTION:
XS GIS Cut Line= 3
      2835370.86     10298863.93      2834502.80     10298343.09
      2833851.73     10298060.96
#Sta/Elev= 30
  4269.1 1266.94  4305.6 1262.93  4320.0 1261.74  4432.3 1250.47  4581.3 1236.50
  4639.0 1231.61  4695.0 1227.32  4741.3 1220.49  4776.6 1219.67  4799.6 1215.66
  4826.9 1214.74  4863.8 1209.09  4885.2 1200.68  4893.2 1193.96  4900.7 1185.39
  4916.3 1178.99  4922.4 1178.49  4937.6 1178.95  4948.3 1175.91  4948.8 1175.41
  4969.7 1175.91  4980.4 1178.42  4996.0 1179.06  5068.1 1179.01  5097.0 1182.67
  5134.0 1195.05  5149.5 1196.47  5235.0 1194.91  5376.4 1195.23  5991.0 1208.06
#Mann=9,-1,0
  4269.1    0.05       0  4305.6    0.12       0  4320.0    0.05       0
  4432.3    0.12       0  4581.3    0.05       0  4639.0    0.12       0
  4922.4    0.05       0  4948.3    0.05       0  4969.7    0.05       0
Bank Sta=4948.3,4969.7
Exp/Cntr=0.3,0.1

Type RM Length L Ch R = 1,59960,509,509,509
BEGIN DESCRIPTION:
LITTLE LLANO RIVER 112.0
END DESCRIPTION:
XS GIS Cut Line= 3
      2835255.71     10298353.13      2834954.50     10298057.00
      2834155.65     10297503.09
#Sta/Elev= 30
  4577.6 1229.31  4581.6 1229.28  4586.2 1228.86  4690.7 1215.44  4761.4 1197.74
  4803.9 1191.50  4825.1 1192.22  4832.2 1188.71  4881.7 1176.93  4913.0 1176.65
  5022.9 1175.84  5026.4 1172.64  5026.9 1172.14  5047.9 1172.64  5095.9 1178.97
  5123.6 1188.40  5138.5 1190.60  5404.0 1196.11  5648.5 1208.39  5684.3 1214.88
  5705.2 1222.62  5735.0 1226.82  5749.8 1232.57  5770.8 1232.88  5800.5 1240.06
  5842.4 1241.74  5878.2 1247.63  5920.5 1260.59  5943.7 1271.38  5972.1 1276.14
#Mann=7,-1,0
  4577.6    0.12       0  4581.6    0.05       0  4586.2    0.12       0
  4913.0    0.05       0  5026.4    0.05       0  5047.9    0.05       0
  5920.5    0.12       0
Bank Sta=5026.4,5047.9
Exp/Cntr=0.3,0.1

Type RM Length L Ch R = 1,59451,917,917,917
BEGIN DESCRIPTION:
LITTLE LLANO RIVER 111.0
END DESCRIPTION:
XS GIS Cut Line= 3
      2835855.67     10298403.09      2835235.75     10297633.00
      2835005.68     10297003.10
#Sta/Elev= 30
  4011.4 1275.00  4147.6 1256.71  4239.3 1247.69  4308.4 1236.07  4334.3 1232.89
  4423.3 1224.17  4509.7 1209.44  4633.3 1201.90  4800.3 1190.77  4850.4 1187.86
  4885.6 1178.32  4972.0 1174.31  4998.0 1169.26  5002.6 1169.26  5004.6 1166.03
  5005.1 1165.53  5026.1 1166.03  5063.8 1171.74  5085.1 1180.64  5106.9 1185.55
  5126.8 1186.09  5141.1 1182.80  5234.1 1191.18  5266.0 1197.10  5304.8 1208.59
  5335.3 1212.95  5473.0 1220.00  5563.7 1233.44  5592.8 1241.71  5670.6 1257.40
#Mann=12,-1,0
  4011.4    0.12       0  4147.6    0.05       0  4308.4    0.12       0
  4334.3    0.05       0  4633.3    0.12       0  4800.3    0.05       0
  4998.0    0.12       0  5004.6    0.07       0  5026.1    0.12       0
  5141.1    0.05       0  5473.0    0.12       0  5592.8    0.05       0
Bank Sta=5004.6,5026.1
Exp/Cntr=0.3,0.1

Type RM Length L Ch R = 1,58534,499,499,499
BEGIN DESCRIPTION:
LITTLE LLANO RIVER 109.0
END DESCRIPTION:
XS GIS Cut Line= 3
      2836655.65     10297503.09      2835836.25     10296945.00
      2835305.68     10296753.11
#Sta/Elev= 30
  4008.6 1351.12  4072.9 1332.81  4087.8 1326.05  4159.7 1303.88  4174.6 1295.53
  4246.4 1268.61  4267.4 1262.99  4282.3 1255.28  4354.2 1234.69  4414.5 1220.99
  4482.9 1207.71  4605.6 1192.07  4677.4 1187.44  4881.9 1180.76  4922.7 1178.41
  4958.6 1167.17  4983.7 1164.03  4984.2 1163.53  5005.4 1164.03  5043.1 1168.71
  5054.4 1173.13  5117.9 1179.98  5245.2 1189.59  5362.2 1206.99  5406.2 1216.87
  5431.6 1226.16  5462.2 1232.49  5487.6 1240.83  5511.0 1244.26  5564.2 1262.23
#Mann=6,-1,0
  4008.6    0.12       0  4414.5    0.05       0  4881.9    0.12       0
  4983.7    0.07       0  5005.4    0.12       0  5117.9    0.05       0
Bank Sta=4983.7,5005.4
Exp/Cntr=0.3,0.1

Type RM Length L Ch R = 1,58035,590,590,590
BEGIN DESCRIPTION:
LITTLE LLANO RIVER 108.0
END DESCRIPTION:
XS GIS Cut Line= 3
      2836905.68     10296953.11      2836125.00     10296552.00
      2835305.65     10296453.11
#Sta/Elev= 30
  4122.3 1337.29  4330.2 1267.99  4358.4 1255.49  4413.3 1239.21  4435.5 1238.20
  4463.3 1225.30  4524.3 1206.63  4529.9 1207.80  4568.6 1198.95  4624.8 1191.42
  4685.2 1184.40  4791.1 1181.37  4838.5 1180.27  4923.6 1173.99  4962.3 1162.97
  4979.3 1160.48  4979.8 1159.98  5001.0 1160.48  5009.4 1164.33  5033.5 1164.40
  5079.9 1171.65  5341.8 1190.85  5412.3 1202.98  5488.1 1210.40  5513.0 1211.88
  5592.1 1226.97  5700.6 1247.94  5744.7 1252.77  5805.1 1266.73  5825.3 1268.89
#Mann=9,-1,0
  4122.3    0.12       0  4624.8    0.05       0  4791.1    0.12       0
  4838.5    0.05       0  4979.3    0.05       0  5001.0    0.05       0
  5488.1    0.12       0  5592.1    0.05       0  5700.6    0.12       0
Bank Sta=4979.3,5001
Exp/Cntr=0.3,0.1

Type RM Length L Ch R = 1,57445,511,511,511
BEGIN DESCRIPTION:
LITTLE LLANO RIVER 107.0
END DESCRIPTION:
XS GIS Cut Line= 3
      2836905.69     10296403.11      2836145.50     10295965.00
      2835405.72     10296353.09
#Sta/Elev= 30
  4122.6 1290.06  4210.9 1271.41  4275.6 1263.09  4284.2 1259.48  4291.4 1244.79
  4297.2 1241.55  4307.2 1225.48  4318.8 1213.72  4328.7 1208.87  4341.9 1197.90
  4371.8 1183.61  4458.1 1177.00  4558.2 1176.41  4715.2 1176.24  4879.4 1170.77
  4919.2 1169.30  4950.8 1160.77  4978.1 1159.29  4986.2 1156.21  4986.7 1155.71
  5007.9 1156.21  5011.7 1159.03  5050.2 1160.63  5078.8 1168.82  5094.7 1169.98
  5502.0 1203.67  5606.7 1217.87  5634.4 1219.39  5688.1 1228.10  5835.4 1252.48
#Mann=7,-1,0
  4122.6    0.12       0  4558.2    0.05       0  4879.4    0.12       0
  4986.2    0.07       0  5007.9    0.12       0  5094.7    0.05       0
  5688.1    0.12       0
Bank Sta=4986.2,5007.9
Exp/Cntr=0.3,0.1

Type RM Length L Ch R = 1,56934,508,508,508
BEGIN DESCRIPTION:
LITTLE LLANO RIVER 106.0
END DESCRIPTION:
XS GIS Cut Line= 3
      2836905.67     10296253.10      2836083.00     10295458.00
      2835505.67     10295153.10
#Sta/Elev= 30
  3855.9 1273.87  3919.5 1260.77  3940.6 1252.35  3954.8 1233.24  3962.0 1227.32
  3983.1 1216.98  4004.4 1200.74  4018.6 1195.02  4046.9 1186.07  4099.8 1178.93
  4141.0 1176.44  4231.7 1175.39  4831.8 1171.69  4888.3 1167.40  4938.0 1158.09
  4987.3 1155.82  4987.8 1155.32  5012.6 1155.82  5053.5 1156.83  5127.6 1167.96
  5237.5 1175.72  5291.0 1190.96  5325.8 1206.38  5402.5 1223.92  5505.9 1254.48
  5573.0 1285.31  5595.0 1297.77  5607.6 1310.84  5617.0 1316.96  5652.9 1326.81
#Mann=7,-1,0
  3855.9    0.12       0  4099.8    0.05       0  4141.0    0.12       0
  4231.7    0.05       0  4987.3    0.05       0  5012.6    0.05       0
  5237.5    0.12       0
Bank Sta=4987.3,5012.6
Exp/Cntr=0.3,0.1

Type RM Length L Ch R = 1,56426,513,513,513
BEGIN DESCRIPTION:
LITTLE LLANO RIVER 105.0
END DESCRIPTION:
XS GIS Cut Line= 3
      2837155.68     10295903.10      2836378.00     10295083.00
      2835705.65     10294903.10
#Sta/Elev= 30
  3869.8 1284.59  3940.4 1275.16  4025.3 1244.96  4075.1 1238.53  4103.4 1226.66
  4124.4 1204.75  4145.5 1189.76  4175.6 1183.05  4188.0 1181.79  4237.7 1174.63
  4280.2 1176.21  4313.0 1171.81  4329.1 1171.19  4435.5 1170.16  4492.1 1178.15
  4520.5 1167.86  4611.3 1161.73  5020.8 1149.26  5021.3 1148.76  5046.1 1149.26
  5100.8 1153.68  5110.8 1155.64  5201.9 1168.77  5253.5 1177.29  5328.5 1199.45
  5379.1 1204.04  5483.5 1221.79  5546.1 1246.11  5567.1 1252.46  5696.0 1296.31
#Mann=14,-1,0
  3869.8    0.12       0  4175.6    0.05       0  4188.0    0.12       0
  4313.0    0.05       0  4329.1    0.12       0  4611.3    0.05       0
  5020.8    0.05       0  5046.1    0.05       0  5100.8    0.12       0
  5110.8    0.05       0  5201.9    0.12       0  5379.1    0.05       0
  5546.1    0.12       0  5567.1    0.05       0
Bank Sta=5020.8,5046.1
Exp/Cntr=0.3,0.1

Type RM Length L Ch R = 1,55913,512,512,512
BEGIN DESCRIPTION:
LITTLE LLANO RIVER 104.0
END DESCRIPTION:
XS GIS Cut Line= 3
      2837405.70     10295403.13      2836610.75     10294628.00
      2835805.67     10294803.11
#Sta/Elev= 30
  3889.7 1281.92  3960.4 1268.68  4192.3 1211.38  4292.9 1194.05  4434.3 1178.40
  4888.0 1156.15  4910.3 1151.56  4943.4 1145.94  4992.3 1144.96  4992.8 1144.46
  5018.6 1144.96  5076.8 1146.83  5098.5 1149.99  5137.4 1163.38  5168.9 1166.02
  5271.3 1166.76  5476.0 1179.65  5520.0 1185.06  5595.2 1201.01  5662.2 1219.19
  5680.6 1227.11  5701.1 1230.59  5706.2 1234.44  5711.4 1232.87  5751.7 1247.31
  5783.0 1256.45  5799.3 1264.68  5804.5 1262.95  5817.3 1268.24  5823.9 1270.16
#Mann=9,-1,0
  3889.7    0.12       0  4192.3    0.05       0  4888.0    0.12       0
  4910.3    0.05       0  4992.3    0.05       0  5018.6    0.05       0
  5595.2    0.12       0  5751.7    0.05       0  5817.3    0.12       0
Bank Sta=4992.3,5018.6
Exp/Cntr=0.3,0.1

Type RM Length L Ch R = 1,55401,581,581,581
BEGIN DESCRIPTION:
LITTLE LLANO RIVER 103.0
END DESCRIPTION:
XS GIS Cut Line= 3
      2837555.70     10294403.12      2836760.00     10294138.00
      2836055.66     10293353.09
#Sta/Elev= 30
  4161.3 1208.71  4192.9 1201.94  4225.1 1187.54  4245.7 1181.31  4308.9 1170.68
  4467.1 1163.62  4488.1 1166.47  4582.9 1162.76  4783.3 1161.76  4835.9 1158.01
  4904.6 1148.24  5000.3 1141.51  5000.8 1141.01  5026.9 1141.51  5027.8 1144.16
  5084.6 1144.94  5105.6 1149.28  5162.4 1150.65  5183.3 1154.89  5233.4 1151.98
  5261.8 1146.13  5275.3 1151.15  5339.5 1164.08  5651.3 1184.25  5769.3 1201.94
  5898.7 1235.95  5912.9 1240.26  5927.1 1249.54  5976.4 1260.76  6054.6 1285.79
#Mann=5,-1,0
  4161.3    0.12       0  4225.1    0.05       0  5000.3    0.03       0
  5026.9    0.05       0  5769.3    0.12       0
Bank Sta=5000.3,5026.9
Exp/Cntr=0.3,0.1

Type RM Length L Ch R = 1,54820,510,510,510
BEGIN DESCRIPTION:
LITTLE LLANO RIVER 102.0
END DESCRIPTION:
XS GIS Cut Line= 3
      2837705.68     10294303.10      2836905.75     10293576.00
      2836105.66     10293103.10
#Sta/Elev= 30
  3919.0 1229.93  3955.4 1223.51  4032.2 1204.92  4046.4 1198.63  4053.8 1191.63
  4079.6 1184.57  4174.1 1175.19  4209.2 1176.88  4280.2 1170.59  4316.7 1171.56
  4336.8 1170.97  4445.2 1169.46  4527.5 1166.50  4563.3 1160.24  4643.3 1159.94
  4676.1 1159.85  4712.0 1165.83  4754.5 1156.40  4938.3 1145.23  4984.9 1136.50
  4985.4 1136.00  5012.0 1136.50  5117.9 1155.22  5389.1 1173.71  5411.9 1178.60
  5586.1 1222.83  5601.7 1231.52  5644.6 1242.66  5724.5 1272.60  5929.4 1331.14
#Mann=10,-1,0
  3919.0    0.05       0  3955.4    0.12       0  4079.6    0.05       0
  4316.7    0.12       0  4336.8    0.05       0  4445.2    0.12       0
  4643.3    0.05       0  4984.9    0.05       0  5012.0    0.05       0
  5411.9    0.12       0
Bank Sta=4984.9,5012
Exp/Cntr=0.3,0.1

Type RM Length L Ch R = 1,54310,511,511,511
BEGIN DESCRIPTION:
LITTLE LLANO RIVER 101.0
END DESCRIPTION:
XS GIS Cut Line= 3
      2837855.71     10293753.13      2837044.75     10293086.00
      2836255.69     10293003.11
#Sta/Elev= 30
  3949.9 1223.38  3985.8 1219.95  3990.8 1220.87  4035.3 1207.23  4084.8 1204.42
  4113.5 1200.41  4271.5 1186.23  4475.8 1167.58  4609.4 1160.96  4881.1 1151.35
  4902.0 1144.77  4937.1 1140.66  4945.8 1135.83  4946.3 1135.33  4972.9 1135.83
  5089.6 1140.86  5129.8 1144.44  5180.1 1144.33  5210.2 1151.93  5240.4 1157.11
  5391.2 1167.44  5421.4 1173.53  5482.0 1193.78  5550.6 1218.77  5555.6 1218.26
  5618.0 1239.53  5713.0 1271.64  5741.8 1280.33  5746.9 1280.42  5793.4 1297.22
#Mann=8,-1,0
  3949.9    0.12       0  3990.8    0.05       0  4271.5    0.12       0
  4609.4    0.05       0  4945.8    0.03       0  4972.9    0.05       0
  5482.0    0.12       0  5618.0    0.05       0
Bank Sta=4945.8,4972.9
Exp/Cntr=0.3,0.1

Type RM Length L Ch R = 1,53799,510,510,510
BEGIN DESCRIPTION:
LITTLE LLANO RIVER 100.0
END DESCRIPTION:
XS GIS Cut Line= 3
      2837405.66     10292703.11      2836909.25     10292600.00
      2836255.72     10292203.13
#Sta/Elev= 30
  4493.0 1166.26  4568.2 1159.79  4646.2 1160.97  4697.2 1159.01  4789.2 1148.24
  4863.8 1143.17  4891.3 1138.73  5030.0 1131.34  5030.5 1130.84  5057.3 1131.34
  5059.1 1134.34  5074.4 1135.75  5080.5 1140.32  5086.3 1139.24  5095.9 1143.28
  5117.3 1146.06  5132.8 1145.89  5138.6 1141.11  5144.6 1141.39  5175.4 1148.76
  5261.6 1156.01  5291.7 1166.00  5349.9 1194.66  5370.6 1200.46  5429.3 1219.53
  5556.7 1267.74  5634.8 1298.61  5671.0 1316.21  5708.4 1328.69  5764.6 1349.30
#Mann=6,-1,0
  4493.0    0.05       0  5030.0    0.03       0  5057.3    0.05       0
  5370.6    0.12       0  5556.7    0.05       0  5708.4    0.12       0
Bank Sta=5030,5057.3
Exp/Cntr=0.3,0.1

Type RM Length L Ch R = 1,53289,512,512,512
BEGIN DESCRIPTION:
LITTLE LLANO RIVER 99.0
END DESCRIPTION:
XS GIS Cut Line= 3
      2837355.67     10292503.10      2837086.25     10292177.00
      2836505.73     10292003.13
#Sta/Elev= 30
  4577.0 1159.53  4804.3 1146.08  4903.3 1143.53  4939.8 1135.03  5020.4 1129.70
  5020.9 1129.20  5047.8 1129.70  5052.8 1134.77  5073.7 1147.31  5100.2 1151.61
  5105.4 1154.66  5125.9 1158.96  5138.5 1164.13  5166.4 1169.05  5178.1 1175.11
  5204.7 1181.32  5209.9 1185.26  5243.0 1191.71  5270.9 1194.00  5282.4 1198.52
  5303.3 1199.64  5334.6 1208.65  5355.5 1216.91  5386.8 1225.79  5397.3 1226.32
  5512.1 1260.41  5574.7 1290.73  5589.5 1295.96  5603.4 1304.89  5606.0 1304.89
#Mann=3,-1,0
  4577.0    0.05       0  5020.4    0.05       0  5047.8    0.05       0
Bank Sta=5020.4,5047.8
Exp/Cntr=0.3,0.1

Type RM Length L Ch R = 1,52777,513,513,513
BEGIN DESCRIPTION:
LITTLE LLANO RIVER 98.0
END DESCRIPTION:
XS GIS Cut Line= 3
      2838205.69     10292553.12      2837395.50     10291770.00
      2836605.73     10291703.12
#Sta/Elev= 30
  3873.2 1222.98  3936.9 1206.88  4054.9 1188.09  4092.5 1180.88  4283.4 1166.05
  4552.2 1152.13  4771.4 1144.48  4792.5 1141.52  4820.8 1141.71  4842.1 1137.18
  4870.4 1137.93  4944.0 1132.97  5009.9 1128.86  5010.4 1128.36  5037.3 1128.86
  5040.0 1131.73  5084.0 1134.17  5130.3 1142.20  5182.7 1145.82  5281.5 1161.31
  5377.0 1173.68  5382.0 1171.87  5421.3 1174.83  5496.5 1192.66  5541.7 1208.36
  5577.9 1216.68  5602.0 1224.41  5616.0 1226.56  5622.0 1229.85  5792.6 1271.57
#Mann=9,-1,0
  3873.2    0.12       0  4054.9    0.05       0  4944.0    0.12       0
  5009.9    0.07       0  5037.3    0.12       0  5084.0    0.05       0
  5182.7    0.12       0  5281.5    0.05       0  5577.9    0.12       0
Bank Sta=5009.9,5037.3
Exp/Cntr=0.3,0.1

Type RM Length L Ch R = 1,52264,571,571,571
BEGIN DESCRIPTION:
LITTLE LLANO RIVER 97.0
END DESCRIPTION:
XS GIS Cut Line= 3
      2838505.66     10292153.09      2837694.00     10291357.00
      2836905.64     10291453.12
#Sta/Elev= 30
  3863.1 1251.58  4018.6 1209.65  4133.5 1191.34  4252.0 1174.06  4393.5 1163.56
  4796.5 1142.73  4853.1 1133.23  4916.7 1135.02  4959.1 1129.43  4959.5 1126.63
  4960.0 1126.13  4986.9 1126.63  4987.4 1129.31  4994.5 1129.63  5068.8 1127.83
  5078.9 1129.62  5087.9 1134.53  5092.9 1131.78  5099.0 1136.27  5119.2 1140.58
  5157.8 1140.81  5170.2 1139.54  5371.0 1155.27  5586.5 1175.75  5622.9 1181.87
  5669.4 1194.46  5750.8 1206.66  5758.4 1205.04  5769.5 1206.80  5794.2 1210.81
#Mann=10,-1,0
  3863.1    0.12       0  4133.5    0.05       0  4959.5    0.05       0
  4986.9    0.05       0  5157.8    0.12       0  5170.2    0.05       0
  5586.5    0.12       0  5669.4    0.05       0  5758.4    0.12       0
  5769.5    0.05       0
Bank Sta=4959.5,4986.9
Exp/Cntr=0.3,0.1

Type RM Length L Ch R = 1,51693,505,505,505
BEGIN DESCRIPTION:
LITTLE LLANO RIVER 96.0
END DESCRIPTION:
XS GIS Cut Line= 3
      2838755.70     10291053.11      2837968.25     10290857.00
      2837155.66     10291253.12
#Sta/Elev= 30
  4188.5 1266.72  4211.7 1262.56  4247.9 1251.27  4289.2 1242.83  4322.5 1238.52
  4376.9 1226.57  4454.4 1203.17  4508.0 1192.62  4559.5 1178.24  4622.2 1167.10
  4729.6 1153.17  4858.4 1140.27  4913.8 1137.40  4924.4 1133.63  4940.8 1131.00
  4947.6 1124.37  4948.1 1123.87  4975.2 1124.37  4998.7 1126.44  5073.1 1125.94
  5208.3 1132.30  5214.2 1135.98  5236.5 1138.54  5425.6 1142.30  5551.9 1147.88
  5619.5 1152.04  5687.1 1159.06  5754.7 1160.04  5760.3 1157.90  5904.0 1172.73
#Mann=6,-1,0
  4188.5    0.12       0  4622.2    0.05       0  4729.6    0.12       0
  4924.4    0.05       0  4947.6    0.03       0  4975.2    0.05       0
Bank Sta=4947.6,4975.2
Exp/Cntr=0.3,0.1

Type RM Length L Ch R = 1,51188,513,513,513
BEGIN DESCRIPTION:
LITTLE LLANO RIVER 95.0
END DESCRIPTION:
XS GIS Cut Line= 3
      2838655.71     10289703.09      2837846.75     10290395.00
      2837055.65     10291203.14
#Sta/Elev= 30
  3935.5 1256.14  3999.8 1231.55  4020.6 1226.69  4034.9 1219.84  4063.4 1211.85
  4070.0 1211.93  4106.2 1199.70  4147.9 1192.27  4155.6 1188.83  4190.8 1184.74
  4219.3 1177.28  4257.9 1171.65  4368.6 1164.18  4637.5 1159.14  4814.8 1149.59
  4843.5 1148.59  4899.9 1141.33  4939.1 1129.40  4999.6 1120.58  5000.1 1120.08
  5027.4 1120.58  5027.7 1124.15  5034.8 1125.45  5077.2 1126.66  5133.8 1134.87
  5331.8 1136.38  5452.0 1141.04  5480.3 1139.92  5664.2 1148.90  6130.9 1177.95
#Mann=6,-1,0
  3935.5    0.12       0  4257.9    0.05       0  4814.8    0.12       0
  4939.1    0.05       0  4999.6    0.03       0  5027.4    0.05       0
Bank Sta=4999.6,5027.4
Exp/Cntr=0.3,0.1

Type RM Length L Ch R = 1,50675,510,510,510
BEGIN DESCRIPTION:
LITTLE LLANO RIVER 94.0
END DESCRIPTION:
XS GIS Cut Line= 3
      2837505.68     10289703.11      2837423.25     10290118.00
      2836605.68     10290353.11
#Sta/Elev= 30
  4577.0 1147.15  4658.8 1143.06  4770.7 1134.84  4893.1 1130.03  4944.0 1120.60
  5000.0 1121.30  5007.9 1120.80  5014.7 1118.29  5015.2 1117.79  5042.6 1118.29
  5049.5 1121.37  5068.9 1122.26  5122.3 1130.31  5253.0 1134.73  5382.5 1141.28
  5458.9 1148.36  5544.0 1158.46  5582.3 1164.63  5601.0 1169.94  5616.0 1171.01
  5621.8 1173.99  5688.6 1189.17  5702.2 1193.75  5756.0 1208.54  5761.2 1208.44
  5794.9 1221.37  5800.2 1221.79  5828.6 1230.86  5833.9 1229.89  5850.7 1236.62
#Mann=6,-1,0
  4577.0    0.05       0  5014.7    0.05       0  5042.6    0.05       0
  5458.9    0.12       0  5544.0    0.05       0  5702.2    0.12       0
Bank Sta=5014.7,5042.6
Exp/Cntr=0.3,0.1

Type RM Length L Ch R = 1,50165,508,508,508
BEGIN DESCRIPTION:
LITTLE LLANO RIVER 93.0
END DESCRIPTION:
XS GIS Cut Line= 3
      2837405.64     10289653.13      2836982.25     10289864.00
      2836305.66     10289653.10
#Sta/Elev= 30
  4527.0 1145.52  4530.2 1145.45  4643.0 1136.37  4876.7 1120.53  4915.9 1125.26
  4921.5 1121.73  4951.5 1117.45  5039.7 1114.95  5040.2 1114.45  5067.7 1114.95
  5101.1 1119.40  5118.7 1129.45  5124.0 1127.44  5151.2 1139.79  5189.0 1143.23
  5203.4 1149.37  5216.3 1154.42  5221.5 1153.29  5237.3 1162.87  5291.8 1183.12
  5319.1 1197.66  5356.8 1211.33  5389.3 1229.57  5427.1 1242.48  5509.7 1282.31
  5524.6 1286.20  5557.1 1304.97  5627.4 1331.52  5697.8 1363.39  5708.7 1367.01
#Mann=7,-1,0
  4527.0    0.05       0  4530.2    0.12       0  4643.0    0.05       0
  5039.7    0.05       0  5067.7    0.05       0  5203.4    0.12       0
  5697.8    0.05       0
Bank Sta=5039.7,5067.7
Exp/Cntr=0.3,0.1

Type RM Length L Ch R = 1,49657,511,511,511
BEGIN DESCRIPTION:
LITTLE LLANO RIVER 92.0
END DESCRIPTION:
XS GIS Cut Line= 3
      2837305.68     10289503.11      2836912.75     10289385.00
      2836505.71     10289453.11
#Sta/Elev= 30
  4589.7 1139.22  4611.4 1135.60  4725.4 1130.32  4903.0 1127.89  4952.2 1115.80
  4992.0 1113.75  5000.0 1113.35  5001.5 1111.41  5002.0 1110.91  5029.5 1111.41
  5057.9 1116.78  5068.0 1121.60  5076.3 1128.48  5081.3 1127.35  5098.4 1142.22
  5108.6 1148.41  5128.8 1156.11  5137.0 1161.09  5142.0 1161.22  5169.4 1178.58
  5197.7 1192.93  5202.8 1192.31  5250.5 1215.31  5258.4 1221.37  5263.5 1219.27
  5270.8 1224.31  5319.1 1246.90  5324.2 1246.29  5351.9 1260.62  5412.7 1285.91
#Mann=4,-1,0
  4589.7    0.05       0  4992.0    0.12       0  5001.5    0.07       0
  5029.5    0.12       0
Bank Sta=5001.5,5029.5
Exp/Cntr=0.3,0.1

Type RM Length L Ch R = 1,49146,585,585,585
BEGIN DESCRIPTION:
LITTLE LLANO RIVER 91.0
END DESCRIPTION:
XS GIS Cut Line= 3
      2837455.69     10289303.12      2837089.75     10288916.00
      2836805.69     10288603.11
#Sta/Elev= 30
  4467.3 1141.36  4722.0 1128.11  4835.2 1125.47  4884.6 1125.95  4898.8 1125.00
  4914.5 1121.47  4955.4 1113.65  5005.3 1111.39  5012.1 1110.36  5012.3 1108.70
  5012.8 1108.20  5040.3 1108.70  5040.5 1112.21  5061.4 1126.57  5075.6 1140.36
  5089.8 1150.73  5097.2 1152.89  5104.0 1156.78  5146.5 1171.46  5153.3 1175.55
  5195.9 1191.51  5210.1 1195.50  5217.5 1195.97  5252.6 1209.82  5281.0 1217.47
  5295.2 1222.94  5344.5 1237.62  5380.4 1245.47  5401.3 1252.42  5422.6 1256.56
#Mann=4,-1,0
  4467.3    0.05       0  4914.5    0.12       0  5012.3    0.07       0
  5040.3    0.12       0
Bank Sta=5012.3,5040.3
Exp/Cntr=0.3,0.1

Type RM Length L Ch R = 1,48561,515,515,515
BEGIN DESCRIPTION:
LITTLE LLANO RIVER 90.0
END DESCRIPTION:
XS GIS Cut Line= 3
      2838355.70     10289353.12      2837558.50     10288569.00
      2837055.68     10288453.11
#Sta/Elev= 30
  3881.8 1163.72  3994.9 1149.24  4143.5 1135.58  4228.3 1130.39  4405.1 1125.33
  4878.8 1123.34  4949.5 1111.79  4970.8 1111.12  4977.9 1108.69  4978.4 1108.19
  5006.0 1108.69  5023.4 1110.90  5048.8 1109.98  5096.7 1118.50  5134.2 1122.23
  5218.4 1131.63  5259.4 1140.14  5310.6 1160.44  5315.8 1159.68  5321.0 1161.62
  5331.3 1166.02  5351.8 1179.21  5371.3 1183.66  5406.5 1191.20  5433.9 1201.84
  5449.3 1205.34  5454.4 1208.59  5497.2 1222.83  5505.7 1225.14  5516.0 1224.86
#Mann=5,-1,0
  3881.8    0.05       0  4977.9    0.03       0  5006.0    0.05       0
  5134.2    0.12       0  5371.3    0.05       0
Bank Sta=4977.9,5006
Exp/Cntr=0.3,0.1

Type RM Length L Ch R = 1,48046,408,408,408
BEGIN DESCRIPTION:
LITTLE LLANO RIVER 89.0
END DESCRIPTION:
XS GIS Cut Line= 3
      2838805.66     10288853.09      2838006.50     10288319.00
      2837355.67     10287803.10
#Sta/Elev= 30
  4038.8 1288.22  4067.3 1277.03  4082.3 1263.15  4103.3 1255.65  4118.3 1242.56
  4124.4 1242.87  4154.4 1226.26  4232.5 1199.37  4262.5 1183.01  4334.6 1160.66
  4437.1 1142.88  4588.2 1127.43  4731.0 1120.79  4773.1 1122.59  4832.6 1118.62
  4853.3 1120.97  4890.2 1120.35  4896.2 1116.65  4939.1 1108.03  4939.6 1107.53
  4967.3 1108.03  5047.7 1108.05  5126.2 1119.85  5289.7 1126.97  5430.1 1137.23
  5465.9 1140.56  5549.8 1149.02  5781.0 1172.47  5799.5 1174.71  5830.5 1178.18
#Mann=11,-1,0
  4038.8    0.12       0  4437.1    0.05       0  4588.2    0.12       0
  4853.3    0.05       0  4939.1    0.03       0  4967.3    0.05       0
  5430.1    0.12       0  5465.9    0.05       0  5549.8    0.12       0
  5781.0    0.05       0  5799.5    0.12       0
Bank Sta=4939.1,4967.3
Exp/Cntr=0.3,0.1

Type RM Length L Ch R = 1,47638,513,513,513
BEGIN DESCRIPTION:
LITTLE LLANO RIVER 88.0
END DESCRIPTION:
XS GIS Cut Line= 3
      2838655.65     10288453.08      2838367.75     10288131.00
      2838305.66     10288003.07
#Sta/Elev= 30
  4568.0 1159.46  4575.1 1158.67  4581.8 1155.21  4589.3 1154.72  4596.0 1152.47
  4603.5 1151.55  4610.2 1149.10  4667.0 1139.97  4681.2 1138.83  4709.6 1134.73
  4730.6 1133.01  4752.3 1129.91  4815.8 1125.05  4822.8 1125.06  4836.7 1123.39
  4901.1 1118.39  4907.8 1116.69  4922.0 1109.72  4922.1 1105.50  4922.6 1105.00
  4949.8 1105.00  4950.3 1105.50  4950.4 1107.56  4960.2 1107.93  4971.3 1108.20
  5020.8 1106.54  5053.2 1107.42  5060.4 1111.19  5075.5 1111.71  5142.2 1118.34
#Mann=4,-1,0
  4568.0    0.12       0  4922.1    0.03       0  4950.3    0.12       0
  4960.2    0.05       0
Bank Sta=4922.1,4950.3
Exp/Cntr=0.3,0.1

Type RM Length L Ch R = 1,47125,516,516,516
BEGIN DESCRIPTION:
LITTLE LLANO RIVER 87.0
END DESCRIPTION:
XS GIS Cut Line= 3
      2839355.65     10288403.08      2838808.50     10287868.00
      2838005.67     10287453.10
#Sta/Elev= 30
  4234.7 1439.31  4238.2 1439.31  4241.7 1434.21  4248.7 1434.14  4255.9 1427.21
  4262.9 1425.12  4305.3 1396.06  4340.7 1374.25  4347.7 1373.07  4397.3 1341.59
  4425.6 1327.71  4439.8 1323.82  4482.2 1298.23  4510.5 1293.96  4545.8 1271.49
  4687.2 1204.33  4729.6 1178.58  4750.9 1175.85  4772.1 1165.23  4821.7 1153.43
  4885.2 1127.79  4913.5 1123.67  4956.0 1101.75  4956.5 1101.25  4984.2 1101.75
  4998.4 1105.83  5081.6 1106.52  5138.2 1114.61  5509.7 1118.94  5903.7 1138.33
#Mann=3,-1,0
  4234.7    0.12       0  4956.0    0.03       0  4984.2    0.05       0
Bank Sta=4956,4984.2
Exp/Cntr=0.3,0.1

Type RM Length L Ch R = 1,46609,517,517,517
BEGIN DESCRIPTION:
LITTLE LLANO RIVER 86.0
END DESCRIPTION:
XS GIS Cut Line= 3
      2839655.68     10288253.11      2838899.00     10287451.00
      2838205.68     10287353.11
#Sta/Elev= 30
  3897.3 1351.36  3918.5 1336.46  3961.0 1319.52  4081.2 1298.38  4152.0 1280.84
  4173.0 1283.79  4251.1 1259.48  4272.1 1259.64  4378.5 1238.66  4491.4 1203.04
  4612.0 1141.32  4689.6 1121.54  4718.0 1102.44  4760.4 1101.13  4771.5 1104.89
  4788.8 1111.96  4795.6 1107.48  4802.9 1113.00  4809.8 1102.71  4817.1 1105.73
  4824.0 1101.44  4866.4 1102.31  4880.6 1108.14  4915.8 1101.91  4999.3 1098.50
  4999.8 1098.00  5027.6 1098.50  5144.7 1114.71  5437.6 1116.84  5700.2 1131.71
#Mann=4,-1,0
  3897.3    0.12       0  4771.5    0.05       0  4999.3    0.03       0
  5027.6    0.05       0
Bank Sta=4999.3,5027.6
Exp/Cntr=0.3,0.1

Type RM Length L Ch R = 1,46092,409,409,409
BEGIN DESCRIPTION:
LITTLE LLANO RIVER 85.0
END DESCRIPTION:
XS GIS Cut Line= 3
      2839455.64     10287103.11      2838662.75     10286993.00
      2838305.67     10286603.10
#Sta/Elev= 30
  4199.5 1170.29  4229.7 1168.17  4280.2 1153.97  4300.4 1134.82  4304.1 1129.68
  4307.0 1125.66  4312.0 1124.24  4330.7 1122.79  4755.5 1114.85  4860.5 1111.52
  4896.1 1110.86  4946.6 1099.24  4948.1 1095.93  4948.6 1095.43  4976.4 1095.93
  5004.8 1098.16  5047.4 1097.15  5082.8 1099.85  5104.1 1100.11  5132.5 1103.21
  5196.0 1113.65  5217.0 1115.33  5255.1 1115.08  5287.9 1111.51  5302.1 1102.75
  5309.5 1101.38  5373.0 1111.51  5408.1 1114.60  5458.1 1125.19  5528.7 1132.12
#Mann=8,-1,0
  4199.5    0.12       0  4304.1    0.05       0  4755.5    0.12       0
  4860.5    0.05       0  4948.1    0.07       0  4976.4    0.05       0
  5082.8    0.05       0  5255.1    0.12       0
Bank Sta=4948.1,4976.4
Exp/Cntr=0.3,0.1

Type RM Length L Ch R = 1,45683,503,503,503
BEGIN DESCRIPTION:
LITTLE LLANO RIVER 84.0
END DESCRIPTION:
XS GIS Cut Line= 3
      2838855.65     10286703.08      2838767.00     10286624.00
      2838655.66     10286553.10
#Sta/Elev= 30
  4881.2 1112.83  4888.3 1112.84  4895.0 1111.67  4902.5 1109.50  4912.3 1105.57
  4923.4 1101.31  4930.9 1097.60  4945.1 1096.13  4959.3 1095.60  4965.8 1093.26
  4966.3 1092.76  4994.1 1092.76  4994.6 1093.26  4997.5 1094.31  5009.2 1094.77
  5015.2 1094.08  5024.5 1095.70  5030.4 1095.65  5037.1 1096.21  5045.6 1097.55
  5060.8 1100.72  5066.8 1102.50  5082.0 1104.36  5088.0 1106.40  5096.4 1106.42
  5103.2 1108.19  5118.4 1111.02  5124.4 1110.79  5129.0 1112.27  5132.0 1112.27
#Mann=4,-1,0
  4881.2    0.05       0  4912.3    0.12       0  4965.8    0.07       0
  4994.6    0.12       0
Bank Sta=4965.8,4994.6
Exp/Cntr=0.3,0.1

Type RM Length L Ch R = 1,45180,509,509,509
BEGIN DESCRIPTION:
LITTLE LLANO RIVER 83.0
END DESCRIPTION:
XS GIS Cut Line= 3
      2839905.67     10287053.10      2839093.25     10286243.00
      2838605.71     10285953.13
#Sta/Elev= 30
  3852.7 1243.36  3923.4 1224.44  4001.2 1209.66  4050.7 1202.41  4149.7 1178.48
  4248.7 1162.70  4284.0 1162.88  4305.2 1165.13  4390.1 1160.66  4411.3 1155.30
  4460.8 1149.14  4496.2 1139.86  4538.6 1133.99  4588.1 1134.49  4715.3 1116.88
  4899.2 1106.59  4920.4 1100.52  4955.8 1094.11  4962.5 1089.78  4963.0 1089.28
  4991.4 1089.78  4996.4 1093.09  5012.1 1091.32  5055.3 1092.89  5129.0 1107.88
  5181.9 1109.67  5325.7 1113.85  5427.5 1119.99  5544.0 1134.38  5567.2 1135.70
#Mann=5,-1,0
  3852.7    0.12       0  4962.5    0.07       0  4991.4    0.12       0
  5181.9    0.05       0  5427.5    0.12       0
Bank Sta=4962.5,4991.4
Exp/Cntr=0.3,0.1

Type RM Length L Ch R = 1,44671,517,517,517
BEGIN DESCRIPTION:
LITTLE LLANO RIVER 82.0
END DESCRIPTION:
XS GIS Cut Line= 3
      2839755.69     10286553.12      2839166.25     10285753.00
      2838705.66     10285653.11
#Sta/Elev= 30
  4006.2 1179.04  4134.6 1161.44  4163.9 1155.84  4249.5 1145.51  4364.5 1138.60
  4414.6 1132.03  4521.1 1122.98  4627.5 1110.86  4821.8 1099.40  4836.5 1098.41
  4842.7 1096.51  4857.3 1097.03  4878.2 1091.54  4913.7 1090.10  4928.3 1091.25
  4978.4 1088.64  5010.8 1089.30  5027.1 1087.71  5027.6 1087.21  5056.0 1087.71
  5073.8 1094.20  5092.7 1103.17  5112.7 1106.75  5215.1 1111.08  5246.2 1112.65
  5266.6 1111.87  5337.1 1116.82  5379.2 1119.53  5430.3 1131.65  5471.3 1135.33
#Mann=5,-1,0
  4006.2    0.12       0  5027.1    0.07       0  5056.0    0.12       0
  5215.1    0.05       0  5337.1    0.12       0
Bank Sta=5027.1,5056
Exp/Cntr=0.3,0.1

Type RM Length L Ch R = 1,44154,507,507,507
BEGIN DESCRIPTION:
LITTLE LLANO RIVER 81.0
END DESCRIPTION:
XS GIS Cut Line= 3
      2839655.71     10285403.12      2839280.75     10285253.00
      2838905.69     10285103.11
#Sta/Elev= 30
  4596.1 1112.35  4800.1 1106.60  4909.7 1102.52  4919.3 1101.10  4928.6 1097.03
  4933.9 1095.82  4940.8 1092.04  4958.2 1087.18  4973.1 1085.48  4980.1 1082.73
  4980.6 1082.23  5009.1 1082.73  5041.6 1087.49  5059.3 1094.67  5065.9 1098.70
  5080.8 1100.94  5090.1 1103.59  5095.5 1103.59  5102.4 1105.55  5119.7 1108.19
  5167.0 1110.21  5197.9 1113.14  5227.5 1119.80  5274.7 1125.98  5296.2 1130.44
  5311.0 1132.50  5328.5 1133.19  5362.0 1136.68  5364.9 1136.45  5403.9 1141.39
#Mann=5,-1,0
  4596.1    0.05       0  4800.1    0.12       0  4980.1    0.07       0
  5009.1    0.12       0  5362.0    0.05       0
Bank Sta=4980.1,5009.1
Exp/Cntr=0.3,0.1

Type RM Length L Ch R = 1,43647,510,510,510
BEGIN DESCRIPTION:
LITTLE LLANO RIVER 80.0
END DESCRIPTION:
XS GIS Cut Line= 3
      2840055.68     10285353.10      2839517.00     10284805.00
      2839055.71     10284753.11
#Sta/Elev= 30
  4231.5 1131.71  4266.8 1128.91  4333.7 1114.13  4449.2 1110.89  4578.0 1108.99
  4853.8 1100.86  4924.5 1093.34  4945.7 1087.97  4952.8 1085.05  4966.9 1082.77
  4981.0 1083.96  4983.3 1081.97  4983.8 1081.47  5012.4 1081.97  5021.5 1082.92
  5031.5 1082.42  5041.6 1084.57  5059.1 1085.95  5081.8 1094.40  5112.0 1102.29
  5134.3 1106.35  5172.4 1109.21  5192.5 1107.11  5212.6 1106.89  5313.3 1111.70
  5329.2 1114.31  5373.7 1117.90  5419.2 1126.67  5454.2 1130.99  5464.2 1133.24
#Mann=6,-1,0
  4231.5    0.12       0  4333.7    0.05       0  4449.2    0.12       0
  4983.3    0.07       0  5012.4    0.12       0  5134.3    0.05       0
Bank Sta=4983.3,5012.4
Exp/Cntr=0.3,0.1

Type RM Length L Ch R = 1,43137,565,565,565
BEGIN DESCRIPTION:
LITTLE LLANO RIVER 79.0
END DESCRIPTION:
XS GIS Cut Line= 3
      2840055.68     10284753.11      2839732.25     10284343.00
      2839105.73     10284353.11
#Sta/Elev= 30
  4477.7 1108.09  4722.1 1102.05  4762.3 1101.70  4797.5 1099.68  4820.0 1100.08
  4840.9 1097.89  4861.7 1093.26  4869.7 1092.96  4919.4 1087.29  4925.8 1085.33
  4948.3 1083.99  4954.7 1082.58  4961.7 1083.04  5011.9 1082.31  5012.4 1081.81
  5040.8 1081.81  5041.3 1082.31  5046.6 1083.59  5086.6 1086.16  5218.4 1091.62
  5296.6 1098.41  5314.2 1101.18  5319.2 1101.18  5326.6 1103.30  5356.6 1107.02
  5436.6 1112.96  5466.6 1117.52  5506.6 1121.03  5556.6 1127.19  5626.6 1133.07
#Mann=5,-1,0
  4477.7    0.05       0  4722.1    0.12       0  5011.9    0.07       0
  5041.3    0.12       0  5218.4    0.12       0
Bank Sta=5011.9,5041.3
Exp/Cntr=0.3,0.1

Type RM Length L Ch R = 1,42572,377,377,377
BEGIN DESCRIPTION:
LITTLE LLANO RIVER 78.0
END DESCRIPTION:
XS GIS Cut Line= 3
      2840405.68     10283253.12      2839867.25     10283795.00
      2839155.65     10284303.14
#Sta/Elev= 30
  4236.1 1133.26  4271.4 1128.06  4328.0 1122.76  4393.3 1120.85  4518.9 1112.31
  4688.6 1095.11  4745.2 1092.89  4872.5 1091.99  4893.7 1087.95  4900.8 1083.99
  4910.6 1083.02  4922.0 1082.99  4936.1 1085.78  4943.2 1085.13  4949.6 1081.59
  4950.1 1081.09  4979.3 1081.59  5031.1 1082.03  5048.8 1082.53  5199.7 1082.32
  5235.4 1086.17  5363.3 1086.73  5401.2 1089.06  5416.0 1094.50  5422.1 1093.11
  5457.7 1098.71  5608.9 1108.13  5709.7 1118.31  5831.3 1125.11  5874.4 1129.42
#Mann=8,-1,0
  4236.1    0.05       0  4393.3    0.12       0  4910.6    0.05       0
  4949.6    0.03       0  4979.3    0.05       0  5031.1    0.12       0
  5048.8    0.05       0  5363.3    0.12       0
Bank Sta=4949.6,4979.3
Exp/Cntr=0.3,0.1

Type RM Length L Ch R = 1,42195,587,587,587
BEGIN DESCRIPTION:
LITTLE LLANO RIVER 77.0
END DESCRIPTION:
XS GIS Cut Line= 3
      2839955.67     10283253.13      2839727.75     10283489.00
      2839405.67     10283803.13
#Sta/Elev= 30
  4672.0 1107.79  4735.6 1098.48  4756.7 1093.85  4763.9 1093.06  4770.9 1091.00
  4785.0 1089.18  4813.3 1087.37  4820.5 1087.78  4955.2 1084.48  4976.2 1083.97
  4996.6 1077.16  4997.1 1076.66  5026.3 1077.16  5032.6 1078.16  5046.7 1077.77
  5075.0 1080.94  5096.3 1081.21  5121.6 1082.85  5138.8 1083.51  5188.2 1081.13
  5244.8 1084.07  5265.6 1086.12  5273.1 1086.25  5315.5 1092.10  5351.0 1093.61
  5365.1 1095.63  5386.2 1096.49  5428.7 1100.89  5435.8 1100.55  5449.9 1101.63
#Mann=6,-1,0
  4672.0    0.12       0  4955.2    0.05       0  4996.6    0.05       0
  5026.3    0.05       0  5121.6    0.12       0  5265.6    0.05       0
Bank Sta=4996.6,5026.3
Exp/Cntr=0.3,0.1

Type RM Length L Ch R = 1,41608,591,591,591
BEGIN DESCRIPTION:
LITTLE LLANO RIVER 76.0
END DESCRIPTION:
XS GIS Cut Line= 3
      2840005.73     10283103.13      2839600.25     10282968.00
      2839255.67     10282753.10
#Sta/Elev= 30
  4572.6 1111.34  4583.2 1111.05  4619.0 1104.15  4646.4 1100.68  4688.6 1091.30
  4798.3 1084.15  4846.7 1083.35  4873.1 1080.39  4899.4 1079.89  4936.3 1075.44
  4983.7 1073.12  4984.7 1071.16  4985.2 1070.66  5014.5 1071.16  5026.4 1071.73
  5042.1 1071.82  5057.4 1074.45  5072.8 1081.34  5078.7 1080.62  5094.0 1085.22
  5123.2 1085.26  5188.4 1088.96  5198.6 1088.54  5209.2 1088.49  5225.0 1090.04
  5230.9 1088.45  5240.3 1090.60  5267.5 1092.77  5377.2 1110.75  5406.1 1112.30
#Mann=8,-1,0
  4572.6    0.05       0  4619.0    0.12       0  4798.3    0.05       0
  4984.7    0.05       0  5014.5    0.05       0  5026.4    0.12       0
  5198.6    0.05       0  5209.2    0.12       0
Bank Sta=4984.7,5014.5
Exp/Cntr=0.3,0.1

Type RM Length L Ch R = 1,41017,511,511,511
BEGIN DESCRIPTION:
Mapping XS b80c3cfd
END DESCRIPTION:
XS GIS Cut Line= 4
      2841208.49     10282826.59      2840514.08     10282652.99
      2839646.02     10282479.38      2839255.38     10282566.19
#Sta/Elev= 30
  3708.7 1115.95  3806.3 1115.25  3876.5 1115.49  3984.0 1110.56  4034.3 1104.13
  4165.1 1094.90  4235.3 1091.08  4405.7 1086.75  4444.1 1085.84  4473.8 1081.41
  4499.8 1083.78  4568.3 1084.53  4682.4 1083.12  4749.2 1080.58  4761.1 1078.37
  4856.8 1075.61  4912.9 1069.45  4989.2 1066.94  4989.7 1066.44  5019.1 1066.94
  5024.5 1068.79  5136.7 1075.76  5167.8 1080.31  5241.1 1084.26  5299.9 1087.57
  5361.3 1093.91  5474.0 1096.87  5531.3 1100.47  5660.1 1108.09  5709.9 1111.03
#Mann=13,-1,0
  3708.7    0.12       0  3806.3    0.05       0  3984.0    0.12       0
  4405.7    0.05       0  4444.1    0.12       0  4568.3    0.05       0
  4682.4    0.12       0  4761.1    0.05       0  4989.2    0.03       0
  5019.1    0.05       0  5241.1    0.12       0  5531.3    0.05       0
  5660.1    0.12       0
Bank Sta=4989.2,5019.1
Exp/Cntr=0.3,0.1
