--- MILLER CREEK.prj (project) ---

Proj Title=MILLER CREEK Base Level Engineering
Current Plan=p01
Default Exp/Contr=0.3,0.1
English Units
Geom File=g01
Flow File=f01
Plan File=p01
BEGIN DESCRIPTION:
MILLER CREEK
END DESCRIPTION:

--- MILLER CREEK.p01 (plan) ---

Plan Title=Multiple Run
Short Identifier=Multiple
Geom File=g01
Flow File=f01
Subcritical Flow
K Sum by GR= 0
Std Step Tol= 0.01
Critical Tol= 0.01
Num of Std Step Trials= 20
Max Error Tol= 0.3
Flow Tol Ratio= 0.001
Split Flow NTrial= 30
Split Flow Tol= 0.02
Split Flow Ratio= 0.02
Log Output Level= 0
Friction Slope Method= 1
Unsteady Friction Slope Method= 2
Unsteady Bridges Friction Slope Method= 1
Parabolic Critical Depth
Global Vel Dist=  1 , 1 , 1
Global Log Level= 0
CheckData=True
Encroach Param= -1, 0, 0, 0
BEGIN DESCRIPTION:
Multiple Run
END DESCRIPTION:

--- MILLER CREEK.f01 (steady flow) ---

Flow Title=Multiple
Number of Profiles=7
Profile Names=10-year,25-year,50-year,1pct_min,100-year,1pct_plu,500-year
River Rch & RM= MILLER CREEK,Reach-1,63783
      69     130     201     104     313     946     822
River Rch & RM= MILLER CREEK,Reach-1,57697
     109     221     354     188     567    1713    1556
River Rch & RM= MILLER CREEK,Reach-1,51213
     145     304     496     267     805    2431    2260
River Rch & RM= MILLER CREEK,Reach-1,47911
     173     374     616     334    1009    3046    2873
River Rch & RM= MILLER CREEK,Reach-1,37600
     203     444     737     402    1214    3666    3496
River Rch & RM= MILLER CREEK,Reach-1,28136
     222     490     817     447    1350    4077    3912
River Rch & RM= MILLER CREEK,Reach-1,19858
     279     626    1054     580    1753    5293    5148
River Rch & RM= MILLER CREEK,Reach-1,17373
     316     715    1208     668    2017    6092    5967
River Rch & RM= MILLER CREEK,Reach-1,9874
     359     818    1388     770    2326    7026    6929
River Rch & RM= MILLER CREEK,Reach-1,7643
     465    1075    1839    1027    3103    9370    9363
River Rch & RM= MILLER CREEK,Reach-1,4757
     484    1122    1921    1074    3244    9797    9808
Boundary for River Rch & Prof#=MILLER CREEK,Reach-1,1
Up Type=0
Dn Type=3
Dn Slope=0.005
Boundary for River Rch & Prof#=MILLER CREEK,Reach-1,2
Up Type=0
Dn Type=3
Dn Slope=0.005
Boundary for River Rch & Prof#=MILLER CREEK,Reach-1,3
Up Type=0
Dn Type=3
Dn Slope=0.005
Boundary for River Rch & Prof#=MILLER CREEK,Reach-1,4
Up Type=0
Dn Type=3
Dn Slope=0.005
Boundary for River Rch & Prof#=MILLER CREEK,Reach-1,5
Up Type=0
Dn Type=3
Dn Slope=0.005
Boundary for River Rch & Prof#=MILLER CREEK,Reach-1,6
Up Type=0
Dn Type=3
Dn Slope=0.005
Boundary for River Rch & Prof#=MILLER CREEK,Reach-1,7
Up Type=0
Dn Type=3
Dn Slope=0.005

--- MILLER CREEK.g01 (geometry) ---

Geom Title=Existing Conditions

River Reach=MILLER CREEK,Reach-1
Reach XY= 30
      2860165.50     10286894.00      2859594.00     10286484.00
      2859622.50     10285024.00      2861124.75     10283908.00
      2862631.50     10280195.00      2863294.00     10280001.00
      2864234.50     10277995.00      2866509.50     10277050.00
      2866225.25     10275513.00      2867312.75     10273179.00
      2866647.00     10272938.00      2866315.75     10270960.00
      2864706.50     10268154.00      2864981.50     10265651.00
      2865375.25     10265382.00      2866231.50     10266170.00
      2866215.75     10263670.00      2866837.75     10262876.00
      2866034.50     10259276.00      2868339.00     10255773.00
      2866065.75     10253526.00      2866350.25     10250991.00
      2865619.00     10250076.00      2863547.00     10249820.00
      2861346.75     10247769.00      2860369.75     10247979.00
      2859614.25     10246337.00      2858526.75     10246559.00
      2858051.75     10246118.00      2857645.50     10244198.00

Type RM Length L Ch R = 1,63783,447,447,447
BEGIN DESCRIPTION:
MILLER CREEK 120.0
END DESCRIPTION:
XS GIS Cut Line= 3
      2860105.65     10286553.12      2859859.50     10286592.00
      2859855.69     10286803.07
#Sta/Elev= 30
  4750.8 1402.93  4760.9 1402.48  4771.0 1401.58  4779.4 1400.47  4784.5 1400.78
  4791.3 1399.85  4841.9 1396.10  4862.1 1395.14  4892.5 1393.16  4902.6 1392.88
  4909.3 1392.22  4937.6 1391.30  4953.2 1390.54  4971.8 1388.99  4976.8 1388.90
  4993.7 1387.72  4997.4 1386.86  4997.7 1386.36  5001.2 1386.36  5001.4 1386.86
  5021.1 1387.19  5031.1 1388.78  5041.1 1389.50  5051.1 1389.29  5061.1 1389.56
  5071.1 1389.16  5100.9 1390.48  5131.1 1392.04  5191.1 1396.68  5211.1 1397.35
#Mann=5,-1,0
  4750.8    0.12       0  4937.6    0.05       0  4997.4    0.05       0
  5001.4    0.05       0  5100.9    0.12       0
Bank Sta=4997.4,5001.4
Exp/Cntr=0.3,0.1

Type RM Length L Ch R = 1,63336,474,474,474
BEGIN DESCRIPTION:
MILLER CREEK 119.0
END DESCRIPTION:
XS GIS Cut Line= 3
      2859905.65     10286403.10      2859592.75     10286331.00
      2859505.71     10286303.12
#Sta/Elev= 30
  4678.9 1391.48  4697.7 1389.85  4702.8 1389.99  4709.7 1388.91  4761.0 1386.58
  4779.1 1385.00  4802.0 1383.89  4812.3 1384.01  4836.3 1382.51  4853.3 1382.75
  4873.8 1382.03  4879.1 1382.50  4894.4 1382.40  4914.9 1381.07  4921.9 1381.44
  4944.3 1380.59  4964.7 1380.22  4993.9 1378.50  4994.2 1378.00  4997.7 1378.00
  4997.9 1378.50  5000.0 1378.50  5005.8 1380.79  5011.1 1381.49  5017.9 1384.16
  5028.4 1387.27  5038.0 1388.83  5043.2 1388.74  5070.1 1393.54  5091.4 1395.05
#Mann=5,-1,0
  4678.9    0.12       0  4779.1    0.05       0  4944.3    0.12       0
  4993.9    0.07       0  4997.9    0.12       0
Bank Sta=4993.9,4997.9
Exp/Cntr=0.3,0.1

Type RM Length L Ch R = 1,62862,465,465,465
BEGIN DESCRIPTION:
MILLER CREEK 118.0
END DESCRIPTION:
XS GIS Cut Line= 3
      2859855.67     10285903.11      2859725.50     10285925.00
      2859455.68     10286003.11
#Sta/Elev= 30
  4868.0 1380.60  4878.1 1379.22  4888.3 1378.73  4895.7 1377.74  4900.8 1378.10
  4918.7 1376.55  4928.8 1376.28  4949.1 1374.34  4956.3 1373.17  4961.4 1373.39
  4979.5 1369.90  4995.4 1369.04  4995.6 1368.54  4999.1 1368.54  4999.4 1369.04
  5002.5 1369.04  5008.1 1370.40  5013.3 1370.86  5041.5 1371.47  5080.5 1373.49
  5119.3 1376.53  5145.6 1380.41  5152.9 1383.14  5158.1 1383.36  5166.4 1385.15
  5176.8 1385.79  5197.6 1388.83  5230.5 1390.53  5264.1 1393.75  5280.9 1395.91
#Mann=3,-1,0
  4868.0    0.12       0  4995.4    0.07       0  4999.4    0.12       0
Bank Sta=4995.4,4999.4
Exp/Cntr=0.3,0.1

Type RM Length L Ch R = 1,62397,380,380,380
BEGIN DESCRIPTION:
MILLER CREEK 117.0
END DESCRIPTION:
XS GIS Cut Line= 3
      2859905.65     10285653.09      2859627.75     10285472.00
      2859455.71     10285553.10
#Sta/Elev= 30
  4668.3 1377.80  4671.2 1377.80  4675.8 1377.00  4681.8 1377.40  4691.0 1375.93
  4696.9 1375.63  4712.0 1372.92  4727.2 1372.03  4739.9 1370.69  4782.3 1368.78
  4805.6 1366.91  4820.7 1366.19  4871.2 1365.06  4893.1 1363.59  4956.4 1364.29
  4978.6 1363.56  4984.7 1362.42  4984.9 1361.92  4988.4 1361.92  4988.7 1362.42
  5003.9 1362.48  5024.4 1365.00  5046.8 1366.31  5062.2 1367.60  5123.9 1370.08
  5130.5 1370.97  5168.1 1372.83  5181.6 1373.97  5187.5 1375.19  5190.2 1375.19
#Mann=5,-1,0
  4668.3    0.12       0  4782.3    0.05       0  4984.7    0.05       0
  4988.7    0.05       0  5046.8    0.12       0
Bank Sta=4984.7,4988.7
Exp/Cntr=0.3,0.1

Type RM Length L Ch R = 1,62017,330,330,330
BEGIN DESCRIPTION:
MILLER CREEK 116.0
END DESCRIPTION:
XS GIS Cut Line= 3
      2859905.66     10285403.08      2859607.00     10285094.00
      2859355.67     10285203.12
#Sta/Elev= 30
  4570.2 1369.08  4605.5 1367.26  4629.8 1365.00  4640.8 1364.05  4654.9 1361.47
  4690.4 1360.73  4747.0 1358.68  4761.2 1358.59  4782.3 1359.54  4824.7 1359.50
  4895.5 1357.67  4937.9 1355.46  4959.2 1356.08  4966.2 1357.32  4994.5 1356.08
  4995.3 1355.18  4995.6 1354.68  4999.1 1354.68  4999.3 1355.18  5014.1 1356.38
  5048.1 1357.70  5107.9 1358.92  5113.3 1359.76  5154.1 1361.22  5165.7 1362.40
  5197.7 1363.35  5207.2 1363.87  5236.1 1367.07  5259.5 1368.13  5274.0 1369.50
#Mann=5,-1,0
  4570.2    0.12       0  4629.8    0.05       0  4995.3    0.05       0
  4999.3    0.05       0  5048.1    0.12       0
Bank Sta=4995.3,4999.3
Exp/Cntr=0.3,0.1

Type RM Length L Ch R = 1,61687,500,500,500
BEGIN DESCRIPTION:
MILLER CREEK 115.0
END DESCRIPTION:
XS GIS Cut Line= 3
      2860105.70     10285453.15      2859798.50     10284869.00
      2859705.69     10284603.13
#Sta/Elev= 30
  4340.0 1380.32  4362.6 1378.03  4407.8 1375.41  4420.0 1373.30  4452.8 1370.41
  4480.5 1370.05  4550.6 1366.58  4590.7 1361.14  4629.1 1357.62  4701.6 1355.56
  4761.4 1355.24  4777.7 1353.82  4814.6 1354.85  4821.8 1353.91  4865.9 1353.21
  4954.1 1353.81  4970.5 1352.51  4992.5 1352.28  5014.8 1347.31  5015.1 1346.81
  5018.8 1347.31  5028.2 1349.91  5038.0 1349.93  5059.3 1355.07  5085.0 1357.56
  5098.9 1359.86  5133.3 1362.84  5141.9 1364.67  5235.0 1377.90  5281.6 1383.36
#Mann=5,-1,0
  4340.0    0.12       0  4550.6    0.05       0  5014.8    0.05       0
  5018.8    0.05       0  5098.9    0.12       0
Bank Sta=5014.8,5018.8
Exp/Cntr=0.3,0.1

Type RM Length L Ch R = 1,61187,433,433,433
BEGIN DESCRIPTION:
MILLER CREEK 114.0
END DESCRIPTION:
XS GIS Cut Line= 3
      2860555.66     10284953.10      2860242.50     10284722.00
      2859955.72     10284453.14
#Sta/Elev= 30
  4610.8 1355.49  4653.6 1352.06  4668.2 1349.92  4724.5 1347.80  4753.8 1344.81
  4789.3 1343.27  4803.9 1345.19  4854.0 1342.87  4918.8 1345.14  4933.4 1344.39
  4939.6 1341.02  4946.3 1342.30  4958.5 1340.84  4958.7 1340.34  4962.5 1340.84
  4975.1 1341.74  4983.6 1344.99  4989.8 1345.50  5000.0 1344.19  5004.1 1341.78
  5018.3 1342.79  5025.1 1344.46  5032.4 1344.18  5039.3 1346.31  5103.2 1348.07
  5130.3 1351.62  5173.8 1358.35  5280.1 1366.86  5357.7 1376.02  5393.1 1379.08
#Mann=4,-1,0
  4610.8    0.05       0  4958.5    0.05       0  4962.5    0.05       0
  5130.3    0.12       0
Bank Sta=4958.5,4962.5
Exp/Cntr=0.3,0.1

Type RM Length L Ch R = 1,60754,480,480,480
BEGIN DESCRIPTION:
MILLER CREEK 113.0
END DESCRIPTION:
XS GIS Cut Line= 3
      2860905.70     10284703.12      2860625.25     10284590.00
      2860355.70     10284403.12
#Sta/Elev= 30
  4697.6 1364.90  4712.4 1363.92  4736.5 1360.12  4751.5 1358.86  4766.1 1356.33
  4814.4 1350.05  4836.3 1347.85  4849.3 1345.71  4891.7 1343.07  4903.0 1341.69
  4986.7 1336.93  4987.0 1336.43  4990.5 1336.43  4990.7 1336.93  5019.3 1337.99
  5040.2 1337.22  5076.0 1337.60  5084.6 1337.80  5090.9 1338.66  5105.8 1338.36
  5133.3 1339.48  5162.5 1341.21  5183.5 1345.34  5206.3 1347.22  5218.9 1350.26
  5234.1 1351.38  5255.1 1354.48  5269.9 1355.41  5305.7 1360.47  5328.0 1362.27
#Mann=5,-1,0
  4697.6    0.12       0  4836.3    0.05       0  4986.7    0.05       0
  4990.7    0.05       0  5218.9    0.12       0
Bank Sta=4986.7,4990.7
Exp/Cntr=0.3,0.1

Type RM Length L Ch R = 1,60274,343,343,343
BEGIN DESCRIPTION:
MILLER CREEK 112.0
END DESCRIPTION:
XS GIS Cut Line= 3
      2861155.69     10284303.12      2860856.75     10284184.00
      2860555.73     10284153.12
#Sta/Elev= 30
  4678.2 1378.65  4693.0 1377.94  4717.3 1370.05  4747.0 1364.53  4753.6 1361.71
  4764.3 1359.72  4795.5 1351.35  4852.6 1339.49  4872.0 1335.75  4893.5 1333.82
  4925.8 1332.92  4938.4 1335.14  4957.3 1331.96  4962.7 1329.70  5009.1 1327.64
  5009.4 1327.14  5013.1 1327.64  5041.3 1329.60  5071.4 1330.26  5091.5 1334.43
  5101.6 1332.96  5111.6 1332.75  5151.3 1335.34  5169.1 1337.49  5192.1 1339.67
  5212.2 1340.00  5250.5 1344.76  5255.5 1344.66  5262.4 1346.55  5302.6 1350.27
#Mann=5,-1,0
  4678.2    0.12       0  4852.6    0.05       0  5009.1    0.05       0
  5013.1    0.05       0  5169.1    0.12       0
Bank Sta=5009.1,5013.1
Exp/Cntr=0.3,0.1

Type RM Length L Ch R = 1,59931,479,479,479
BEGIN DESCRIPTION:
MILLER CREEK 111.0
END DESCRIPTION:
XS GIS Cut Line= 3
      2861155.69     10283953.11      2861100.00     10283943.00
      2860855.64     10283903.10
#Sta/Elev= 30
  4943.4 1336.47  4945.9 1336.47  4953.6 1333.96  4963.7 1330.13  4968.8 1328.59
  4975.2 1324.78  4982.1 1321.99  4982.3 1321.49  4985.8 1321.49  4986.1 1321.99
  4994.2 1322.35  4999.7 1323.71  5004.7 1323.71  5014.5 1325.07  5024.6 1325.41
  5030.0 1325.85  5035.1 1325.90  5055.0 1325.45  5075.3 1326.42  5085.4 1326.62
  5091.4 1327.00  5096.5 1327.03  5115.8 1327.87  5126.0 1328.13  5136.1 1328.88
  5176.6 1329.99  5207.0 1331.73  5227.3 1331.89  5245.0 1332.92  5247.6 1332.92
#Mann=3,-1,0
  4943.4    0.05       0  4982.1    0.05       0  4986.1    0.05       0
Bank Sta=4982.1,4986.1
Exp/Cntr=0.3,0.1

Type RM Length L Ch R = 1,59452,426,426,426
BEGIN DESCRIPTION:
MILLER CREEK 110.0
END DESCRIPTION:
XS GIS Cut Line= 3
      2861405.66     10283803.08      2861205.00     10283519.00
      2861005.73     10283503.12
#Sta/Elev= 30
  4652.2 1339.41  4655.2 1339.41  4659.6 1338.47  4674.3 1337.03  4680.5 1337.08
  4695.3 1335.01  4710.0 1334.06  4737.9 1333.56  4745.7 1331.93  4766.6 1329.60
  4823.6 1326.33  4873.7 1322.57  4884.0 1322.26  4968.6 1319.34  4974.7 1318.56
  4982.7 1315.99  4993.1 1315.83  4993.3 1315.33  4996.8 1315.33  4997.1 1315.83
  5002.2 1315.83  5007.8 1316.93  5019.4 1318.38  5041.5 1319.65  5089.6 1322.39
  5109.7 1322.67  5135.9 1324.41  5140.9 1324.07  5169.9 1325.75  5199.9 1326.80
#Mann=5,-1,0
  4652.2    0.05       0  4884.0    0.12       0  4993.1    0.07       0
  4997.1    0.12       0  5041.5    0.05       0
Bank Sta=4993.1,4997.1
Exp/Cntr=0.3,0.1

Type RM Length L Ch R = 1,59026,345,345,345
BEGIN DESCRIPTION:
MILLER CREEK 109.0
END DESCRIPTION:
XS GIS Cut Line= 3
      2861505.68     10283353.11      2861313.50     10283110.00
      2861005.70     10283153.11
#Sta/Elev= 30
  4690.1 1322.96  4775.9 1319.31  4831.9 1317.83  4860.8 1316.54  4868.6 1316.75
  4889.7 1316.17  4904.1 1316.73  4924.9 1316.50  4945.7 1314.28  4953.8 1314.02
  4968.2 1312.41  4974.6 1311.01  4987.0 1309.86  4987.3 1309.36  4990.8 1309.36
  4991.0 1309.86  5000.0 1310.20  5018.0 1313.41  5038.2 1313.71  5048.3 1313.41
  5068.5 1314.45  5078.6 1313.55  5088.7 1311.53  5098.8 1311.41  5108.9 1312.81
  5149.3 1315.43  5203.7 1317.61  5230.0 1319.19  5275.1 1320.86  5310.8 1323.21
#Mann=3,-1,0
  4690.1    0.05       0  4987.0    0.03       0  4991.0    0.05       0
Bank Sta=4987,4991
Exp/Cntr=0.3,0.1

Type RM Length L Ch R = 1,58681,495,495,495
BEGIN DESCRIPTION:
MILLER CREEK 108.0
END DESCRIPTION:
XS GIS Cut Line= 3
      2861605.71     10283053.15      2861402.75     10282786.00
      2861105.70     10282703.12
#Sta/Elev= 30
  4664.5 1313.57  4771.6 1311.32  4871.5 1310.04  4886.0 1309.47  4921.4 1309.45
  4950.5 1308.53  4956.7 1308.89  4965.0 1307.89  4978.5 1303.90  4990.1 1301.71
  4990.4 1301.21  4993.9 1301.21  4994.1 1301.71  4998.7 1303.17  5026.1 1309.28
  5067.8 1308.34  5099.7 1307.93  5121.5 1308.24  5144.2 1306.88  5163.1 1306.63
  5204.6 1307.08  5212.6 1305.54  5217.8 1305.66  5225.4 1304.25  5235.7 1305.74
  5252.0 1312.06  5266.9 1315.45  5291.3 1318.67  5298.0 1320.52  5308.4 1321.48
#Mann=4,-1,0
  4664.5    0.05       0  4990.1    0.05       0  4994.1    0.05       0
  5067.8    0.12       0
Bank Sta=4990.1,4994.1
Exp/Cntr=0.3,0.1

Type RM Length L Ch R = 1,58186,489,489,489
BEGIN DESCRIPTION:
MILLER CREEK 107.0
END DESCRIPTION:
XS GIS Cut Line= 3
      2861855.68     10283103.11      2861511.50     10282353.00
      2861105.67     10282103.10
#Sta/Elev= 30
  4174.7 1318.58  4234.9 1317.11  4259.7 1315.02  4349.9 1313.33  4526.2 1307.39
  4540.2 1306.85  4581.8 1304.66  4746.6 1300.69  4856.9 1298.98  4860.2 1297.83
  4883.2 1296.57  4906.2 1297.39  4922.9 1296.11  4967.1 1296.35  4973.3 1295.95
  4980.7 1296.47  4995.2 1293.06  4995.4 1292.56  4999.2 1293.06  5026.4 1296.23
  5041.8 1296.91  5053.8 1295.56  5099.1 1298.75  5136.0 1301.34  5200.3 1303.04
  5258.3 1307.38  5374.2 1318.12  5389.6 1321.98  5417.9 1325.54  5476.6 1330.39
#Mann=11,-1,0
  4174.7    0.12       0  4259.7    0.05       0  4526.2    0.12       0
  4540.2    0.05       0  4746.6    0.12       0  4856.9    0.05       0
  4967.1    0.12       0  4973.3    0.05       0  4995.2    0.05       0
  4999.2    0.05       0  5099.1    0.12       0
Bank Sta=4995.2,4999.2
Exp/Cntr=0.3,0.1

Type RM Length L Ch R = 1,57697,378,378,378
BEGIN DESCRIPTION:
MILLER CREEK 106.0
END DESCRIPTION:
XS GIS Cut Line= 3
      2861905.68     10282803.12      2861837.25     10281992.00
      2861505.72     10281603.15
#Sta/Elev= 30
  4186.0 1307.98  4216.1 1307.29  4235.1 1305.85  4296.1 1303.83  4363.0 1301.49
  4386.7 1301.44  4395.0 1300.42  4597.4 1295.07  4790.8 1293.64  4868.4 1292.50
  4918.6 1293.14  4968.8 1291.68  4988.8 1289.53  4996.9 1285.98  5002.6 1285.98
  5007.6 1283.42  5012.2 1282.13  5012.4 1281.63  5016.2 1282.13  5019.3 1282.26
  5036.2 1285.53  5106.4 1291.14  5156.2 1294.07  5192.1 1295.23  5227.2 1297.86
  5319.4 1301.80  5340.3 1304.22  5361.0 1308.16  5405.1 1314.03  5511.0 1322.78
#Mann=9,-1,0
  4186.0    0.12       0  4235.1    0.05       0  4296.1    0.12       0
  4395.0    0.05       0  4790.8    0.12       0  5012.2    0.07       0
  5016.2    0.12       0  5019.3    0.05       0  5361.0    0.12       0
Bank Sta=5012.2,5016.2
Exp/Cntr=0.3,0.1

Type RM Length L Ch R = 1,57319,384,384,384
BEGIN DESCRIPTION:
MILLER CREEK 105.0
END DESCRIPTION:
XS GIS Cut Line= 3
      2862855.68     10281803.11      2862076.00     10281706.00
      2861855.64     10281603.09
#Sta/Elev= 30
  4214.3 1344.29  4252.2 1332.79  4257.2 1335.21  4332.9 1310.83  4337.6 1311.86
  4375.5 1303.81  4413.7 1298.61  4436.6 1297.57  4476.3 1294.36  4526.7 1292.33
  4607.3 1290.94  4729.0 1285.86  4741.8 1285.29  4758.5 1281.10  4778.6 1278.94
  4815.4 1278.87  4815.7 1278.37  4819.5 1278.87  4839.1 1280.25  4939.9 1280.96
  4949.9 1283.08  4960.0 1282.90  4970.1 1280.39  4979.0 1279.68  5011.4 1279.48
  5033.5 1285.19  5077.6 1286.48  5116.7 1289.44  5154.9 1293.68  5243.2 1299.87
#Mann=7,-1,0
  4214.3    0.12       0  4337.6    0.05       0  4436.6    0.12       0
  4729.0    0.05       0  4815.4    0.05       0  4819.5    0.05       0
  5116.7    0.12       0
Bank Sta=4815.4,4819.5
Exp/Cntr=0.3,0.1

Type RM Length L Ch R = 1,56935,461,461,461
BEGIN DESCRIPTION:
MILLER CREEK 104.0
END DESCRIPTION:
XS GIS Cut Line= 3
      2862755.68     10281503.11      2862357.50     10281490.00
      2861955.71     10281503.11
#Sta/Elev= 30
  4601.6 1343.23  4604.1 1343.23  4611.6 1339.48  4632.8 1332.20  4671.6 1318.26
  4681.6 1316.19  4711.7 1308.12  4721.7 1304.40  4750.1 1298.31  4755.1 1298.24
  4821.7 1289.24  4861.7 1285.53  4941.8 1280.14  4951.8 1278.68  4961.8 1278.14
  4981.8 1273.80  4991.8 1272.52  5009.4 1271.99  5009.8 1271.49  5013.9 1271.49
  5014.2 1271.99  5041.8 1275.89  5091.9 1278.62  5131.9 1280.26  5141.9 1279.94
  5181.9 1282.01  5302.0 1284.32  5332.9 1286.10  5362.0 1286.63  5402.0 1289.35
#Mann=5,-1,0
  4601.6    0.12       0  4632.8    0.05       0  5009.4    0.05       0
  5014.2    0.05       0  5332.9    0.12       0
Bank Sta=5009.4,5014.2
Exp/Cntr=0.3,0.1

Type RM Length L Ch R = 1,56474,424,424,424
BEGIN DESCRIPTION:
MILLER CREEK 103.0
END DESCRIPTION:
XS GIS Cut Line= 3
      2862805.66     10281453.09      2862428.75     10281035.00
      2862055.72     10281103.11
#Sta/Elev= 30
  4437.1 1360.49  4444.2 1359.98  4465.1 1351.55  4472.6 1350.77  4479.3 1346.30
  4486.8 1346.80  4493.5 1342.16  4507.7 1337.76  4515.2 1337.47  4529.4 1332.69
  4536.1 1328.72  4557.8 1324.77  4564.5 1321.53  4585.9 1316.09  4592.9 1315.30
  4628.0 1305.04  4672.7 1295.98  4819.3 1278.35  4860.5 1275.24  4918.7 1273.10
  4953.9 1267.80  4961.3 1267.87  4968.1 1264.77  4979.8 1263.84  4980.2 1263.34
  4984.7 1263.84  5057.3 1270.52  5071.1 1272.15  5297.2 1280.80  5379.2 1284.21
#Mann=7,-1,0
  4437.1    0.12       0  4585.9    0.05       0  4860.5    0.12       0
  4979.8    0.07       0  4984.7    0.12       0  5057.3    0.05       0
  5297.2    0.12       0
Bank Sta=4979.8,4984.7
Exp/Cntr=0.3,0.1

Type RM Length L Ch R = 1,56050,494,494,494
BEGIN DESCRIPTION:
MILLER CREEK 102.0
END DESCRIPTION:
XS GIS Cut Line= 3
      2862905.68     10281003.11      2862491.50     10280620.00
      2862205.64     10280703.12
#Sta/Elev= 30
  4435.8 1326.19  4439.2 1326.19  4457.1 1321.09  4463.9 1320.32  4471.2 1317.53
  4513.8 1310.16  4542.1 1302.43  4605.6 1294.17  4619.8 1291.53  4648.1 1288.19
  4697.5 1284.50  4733.2 1279.03  4747.4 1278.76  4761.5 1276.53  4825.0 1270.91
  4860.2 1268.93  4924.3 1267.91  4952.6 1266.11  4966.8 1264.48  4978.2 1260.36
  4978.6 1259.86  4983.1 1260.36  5013.4 1260.96  5047.7 1263.44  5069.3 1263.19
  5120.6 1266.81  5212.8 1270.46  5235.2 1271.33  5256.0 1273.43  5297.7 1275.15
#Mann=5,-1,0
  4435.8    0.12       0  4978.2    0.07       0  4983.1    0.12       0
  5013.4    0.05       0  5212.8    0.12       0
Bank Sta=4978.2,4983.1
Exp/Cntr=0.3,0.1

Type RM Length L Ch R = 1,55556,497,497,497
BEGIN DESCRIPTION:
MILLER CREEK 101.0
END DESCRIPTION:
XS GIS Cut Line= 3
      2862955.68     10280453.11      2862657.25     10280159.00
      2862455.71     10279903.14
#Sta/Elev= 30
  4581.0 1279.61  4665.8 1269.99  4694.1 1267.61  4701.2 1267.78  4708.2 1266.35
  4715.4 1266.64  4736.5 1264.53  4757.8 1263.67  4764.8 1262.37  4786.1 1261.81
  4793.1 1260.43  4807.2 1259.69  4885.1 1257.20  4920.4 1254.81  4969.9 1253.67
  4984.1 1252.58  4991.1 1251.21  4997.6 1248.72  5009.5 1248.69  5010.0 1248.19
  5014.9 1248.69  5026.7 1249.07  5033.2 1250.10  5061.9 1257.62  5105.3 1259.24
  5140.5 1259.39  5169.4 1260.76  5200.9 1264.07  5297.7 1277.40  5325.7 1280.00
#Mann=5,-1,0
  4581.0    0.12       0  5009.5    0.07       0  5014.9    0.12       0
  5033.2    0.05       0  5200.9    0.12       0
Bank Sta=5009.5,5014.9
Exp/Cntr=0.3,0.1

Type RM Length L Ch R = 1,55059,481,481,481
BEGIN DESCRIPTION:
MILLER CREEK 100.0
END DESCRIPTION:
XS GIS Cut Line= 3
      2863205.65     10280203.08      2863122.00     10280123.00
      2863005.68     10280053.11
#Sta/Elev= 30
  4884.2 1253.72  4887.6 1253.72  4905.4 1250.47  4919.5 1242.89  4926.5 1234.74
  4933.7 1230.46  4940.6 1221.88  4947.8 1218.16  4954.8 1211.70  4962.0 1210.06
  4968.9 1206.94  4980.4 1206.52  4980.8 1206.02  4985.4 1206.02  4985.8 1206.52
  4990.3 1208.47  4996.3 1207.30  5000.0 1207.30  5005.5 1210.50  5011.3 1210.00
  5019.0 1213.78  5026.9 1215.08  5042.4 1215.90  5069.6 1222.45  5077.4 1225.92
  5085.2 1230.27  5091.0 1231.10  5100.7 1234.72  5112.4 1237.60  5135.7 1241.11
#Mann=3,-1,0
  4884.2    0.12       0  4980.4    0.07       0  4985.8    0.12       0
Bank Sta=4980.4,4985.8
Exp/Cntr=0.3,0.1

Type RM Length L Ch R = 1,54578,476,476,476
BEGIN DESCRIPTION:
MILLER CREEK 99.0
END DESCRIPTION:
XS GIS Cut Line= 3
      2863505.64     10279803.09      2863397.00     10279763.00
      2863205.66     10279703.10
#Sta/Elev= 30
  4884.2 1225.64  4886.8 1225.64  4894.0 1223.52  4899.4 1222.75  4905.5 1220.73
  4916.1 1218.64  4948.1 1207.78  4954.9 1204.05  4960.2 1201.96  4969.4 1199.54
  4977.3 1198.94  4977.7 1198.44  4982.3 1198.44  4982.7 1198.94  5003.3 1199.81
  5049.2 1206.32  5086.9 1209.37  5106.2 1213.66  5114.1 1216.41  5119.3 1216.38
  5127.1 1219.30  5134.5 1221.25  5146.5 1225.01  5151.8 1225.13  5158.6 1228.25
  5179.0 1234.23  5184.2 1234.72  5190.0 1237.52  5197.9 1240.46  5200.5 1240.46
#Mann=4,-1,0
  4884.2    0.12       0  4977.3    0.07       0  4982.7    0.12       0
  5134.5    0.05       0
Bank Sta=4977.3,4982.7
Exp/Cntr=0.3,0.1

Type RM Length L Ch R = 1,54102,480,480,480
BEGIN DESCRIPTION:
MILLER CREEK 98.0
END DESCRIPTION:
XS GIS Cut Line= 3
      2863705.71     10279453.14      2863597.25     10279332.00
      2863255.67     10279403.11
#Sta/Elev= 30
  4837.4 1202.66  4885.7 1200.96  4915.6 1199.38  4929.8 1197.45  4936.5 1195.39
  4958.2 1192.19  4964.9 1190.53  4979.1 1189.37  4985.8 1185.98  4993.3 1185.83
  4994.7 1185.24  4995.1 1184.74  4999.7 1184.74  5000.2 1185.24  5011.8 1185.32
  5022.0 1186.65  5028.6 1189.60  5033.7 1188.62  5042.5 1191.08  5073.1 1196.28
  5078.6 1197.72  5144.6 1200.35  5162.1 1200.37  5216.1 1203.09  5246.7 1205.64
  5267.2 1208.50  5284.9 1212.33  5318.2 1217.70  5346.3 1225.53  5348.9 1225.53
#Mann=6,-1,0
  4837.4    0.05       0  4885.7    0.12       0  4994.7    0.03       0
  5000.2    0.12       0  5162.1    0.12       0  5284.9    0.05       0
Bank Sta=4994.7,5000.2
Exp/Cntr=0.3,0.1

Type RM Length L Ch R = 1,53622,482,482,482
BEGIN DESCRIPTION:
MILLER CREEK 97.0
END DESCRIPTION:
XS GIS Cut Line= 3
      2863905.68     10279053.11      2863803.25     10278904.00
      2863405.72     10279003.10
#Sta/Elev= 30
  4819.1 1195.76  4819.6 1195.76  4826.5 1195.73  4832.6 1194.90  4847.5 1194.86
  4898.3 1190.55  4904.3 1189.55  4963.9 1186.11  4984.9 1182.22  4997.5 1180.52
  5007.8 1180.50  5015.0 1181.48  5017.2 1180.30  5017.7 1179.80  5022.5 1179.80
  5023.0 1180.30  5028.4 1182.50  5054.4 1189.62  5056.3 1190.21  5061.4 1189.85
  5069.6 1191.99  5079.9 1193.10  5097.5 1194.03  5138.8 1193.95  5144.0 1194.72
  5162.4 1193.90  5317.0 1194.75  5337.6 1196.25  5345.2 1195.63  5409.7 1197.08
#Mann=5,-1,0
  4819.1    0.05       0  4819.6    0.12       0  5017.2    0.07       0
  5023.0    0.12       0  5054.4    0.05       0
Bank Sta=5017.2,5023
Exp/Cntr=0.3,0.1

Type RM Length L Ch R = 1,53140,467,467,467
BEGIN DESCRIPTION:
MILLER CREEK 96.0
END DESCRIPTION:
XS GIS Cut Line= 3
      2864255.72     10278603.13      2864112.75     10278538.00
      2863955.68     10278553.11
#Sta/Elev= 30
  4842.9 1193.73  4845.7 1193.73  4851.7 1193.19  4864.9 1190.90  4880.3 1188.96
  4886.9 1187.54  4897.8 1186.44  4903.3 1186.45  4908.9 1185.23  4919.9 1184.46
  4931.9 1183.04  4944.0 1182.33  4952.1 1181.40  4972.5 1179.01  4978.0 1177.74
  4995.5 1175.23  5004.2 1174.79  5004.6 1174.29  5009.5 1174.29  5010.0 1174.79
  5017.1 1174.99  5027.2 1176.86  5047.3 1179.17  5077.4 1184.06  5087.5 1185.21
  5097.5 1185.54  5104.1 1186.97  5109.1 1186.77  5137.7 1189.66  5157.8 1190.43
#Mann=5,-1,0
  4842.9    0.05       0  4944.0    0.12       0  4952.1    0.05       0
  5004.2    0.03       0  5010.0    0.05       0
Bank Sta=5004.2,5010
Exp/Cntr=0.3,0.1

Type RM Length L Ch R = 1,52673,470,470,470
BEGIN DESCRIPTION:
MILLER CREEK 95.0
END DESCRIPTION:
XS GIS Cut Line= 3
      2864355.68     10278453.11      2864216.00     10278116.00
      2863855.67     10277753.10
#Sta/Elev= 30
  4635.1 1189.56  4712.3 1185.44  4827.8 1179.83  4833.2 1176.19  4840.8 1177.92
  4857.1 1178.23  4862.5 1174.92  4881.0 1176.19  4886.4 1174.12  4904.8 1173.75
  4910.3 1170.46  4934.1 1171.81  4939.6 1169.80  4946.1 1169.56  4946.6 1169.06
  4951.9 1169.56  4987.3 1169.80  4992.7 1171.53  5003.8 1170.92  5009.3 1172.62
  5023.5 1173.46  5065.9 1174.34  5122.5 1172.43  5136.6 1174.72  5157.9 1180.99
  5189.6 1181.60  5249.8 1182.59  5306.3 1186.05  5412.4 1186.09  5511.4 1189.59
#Mann=5,-1,0
  4635.1    0.05       0  4712.3    0.12       0  4946.1    0.07       0
  4951.9    0.12       0  5189.6    0.05       0
Bank Sta=4946.1,4951.9
Exp/Cntr=0.3,0.1

Type RM Length L Ch R = 1,52203,499,499,499
BEGIN DESCRIPTION:
MILLER CREEK 94.0
END DESCRIPTION:
XS GIS Cut Line= 3
      2864455.68     10278253.11      2864528.50     10278123.00
      2864555.68     10278003.14
#Sta/Elev= 30
  4850.9 1182.26  4853.8 1182.26  4858.9 1181.11  4864.6 1178.77  4880.6 1176.64
  4886.3 1174.47  4896.5 1173.56  4902.3 1171.28  4908.2 1170.29  4939.9 1169.14
  4945.7 1168.43  4967.4 1168.57  4977.0 1169.02  4983.3 1168.81  4989.1 1168.31
  4997.1 1166.78  5002.5 1166.78  5007.4 1164.54  5009.7 1164.46  5010.1 1163.96
  5015.0 1163.96  5015.5 1164.46  5020.4 1165.56  5030.6 1166.80  5050.6 1171.29
  5055.7 1170.90  5061.4 1173.13  5071.7 1174.56  5092.2 1174.56  5122.9 1176.41
#Mann=3,-1,0
  4850.9    0.05       0  5009.7    0.03       0  5015.5    0.05       0
Bank Sta=5009.7,5015.5
Exp/Cntr=0.3,0.1

Type RM Length L Ch R = 1,51704,491,491,491
BEGIN DESCRIPTION:
MILLER CREEK 93.0
END DESCRIPTION:
XS GIS Cut Line= 3
      2865055.67     10278553.09      2864828.25     10277954.00
      2864805.68     10277853.09
#Sta/Elev= 30
  4359.2 1178.16  4466.1 1173.49  4484.1 1171.98  4508.9 1172.32  4551.7 1174.72
  4599.3 1173.58  4624.0 1172.11  4722.8 1169.98  4769.4 1166.68  4787.0 1166.17
  4799.5 1164.63  4824.3 1163.63  4837.4 1162.18  4861.9 1161.56  4884.5 1163.28
  4913.1 1162.88  4979.6 1160.29  4989.0 1160.63  4991.4 1158.84  4991.9 1158.34
  4997.4 1158.84  5011.2 1160.21  5021.4 1160.08  5030.6 1161.41  5035.7 1164.19
  5052.1 1170.06  5072.6 1171.21  5079.1 1172.45  5084.2 1174.58  5103.4 1175.27
#Mann=5,-1,0
  4359.2    0.05       0  4837.4    0.12       0  4913.1    0.05       0
  4991.4    0.05       0  4997.4    0.05       0
Bank Sta=4991.4,4997.4
Exp/Cntr=0.3,0.1

Type RM Length L Ch R = 1,51213,476,476,476
BEGIN DESCRIPTION:
MILLER CREEK 92.0
END DESCRIPTION:
XS GIS Cut Line= 3
      2865305.69     10278103.14      2865256.50     10277913.00
      2865005.72     10277703.14
#Sta/Elev= 30
  4803.6 1172.91  4804.4 1172.91  4834.6 1169.62  4867.1 1168.23  4907.8 1164.59
  4937.9 1163.03  4943.2 1163.72  4958.6 1161.85  4968.9 1161.86  4983.8 1159.33
  4989.6 1156.03  4994.3 1154.44  4994.8 1153.94  5000.4 1154.44  5021.9 1156.26
  5028.4 1158.33  5036.2 1157.07  5042.7 1160.18  5050.5 1159.60  5057.1 1161.38
  5079.2 1161.76  5114.3 1164.14  5120.8 1165.58  5127.3 1165.44  5135.1 1166.53
  5142.9 1166.06  5149.4 1167.37  5178.1 1168.20  5221.0 1171.30  5327.0 1172.40
#Mann=5,-1,0
  4803.6    0.05       0  4804.4    0.12       0  4994.3    0.07       0
  5000.4    0.12       0  5127.3    0.05       0
Bank Sta=4994.3,5000.4
Exp/Cntr=0.3,0.1

Type RM Length L Ch R = 1,50737,446,446,446
BEGIN DESCRIPTION:
MILLER CREEK 91.0
END DESCRIPTION:
XS GIS Cut Line= 3
      2865805.67     10277853.10      2865509.50     10277694.00
      2865155.72     10277703.11
#Sta/Elev= 30
  4663.8 1171.48  4799.3 1165.21  4819.6 1163.77  4834.1 1163.66  4841.6 1161.89
  4847.2 1161.36  4863.5 1163.71  4869.2 1163.16  4885.4 1164.31  4891.1 1163.86
  4907.3 1159.94  4913.5 1154.11  4920.5 1152.88  4921.0 1152.38  4926.2 1152.38
  4926.7 1152.88  4929.2 1156.36  4936.2 1153.54  4973.1 1154.54  4981.6 1154.46
  4989.3 1153.49  4995.0 1154.48  4999.3 1153.62  5004.4 1153.62  5023.8 1160.22
  5043.8 1160.86  5143.9 1160.73  5173.9 1161.27  5233.9 1166.27  5353.9 1170.59
#Mann=4,-1,0
  4663.8    0.12       0  4799.3    0.05       0  4920.5    0.05       0
  4926.7    0.05       0
Bank Sta=4920.5,4926.7
Exp/Cntr=0.3,0.1

Type RM Length L Ch R = 1,50291,450,450,450
BEGIN DESCRIPTION:
MILLER CREEK 90.0
END DESCRIPTION:
XS GIS Cut Line= 3
      2865905.68     10277803.10      2865644.00     10277426.00
      2865255.68     10277303.11
#Sta/Elev= 30
  4541.0 1172.23  4641.0 1167.78  4727.4 1165.07  4742.3 1165.29  4748.4 1164.64
  4799.0 1163.85  4864.5 1165.11  4900.0 1164.32  4930.0 1161.72  4965.8 1154.27
  4971.9 1156.80  4992.9 1156.51  4998.7 1151.41  5016.1 1151.19  5016.6 1150.69
  5021.9 1150.69  5022.4 1151.19  5025.3 1151.41  5030.5 1153.63  5040.2 1154.71
  5057.6 1154.81  5062.8 1157.26  5089.9 1159.19  5095.2 1161.72  5113.6 1164.16
  5127.5 1165.01  5154.5 1165.15  5159.8 1165.91  5262.5 1167.58  5407.3 1170.33
#Mann=5,-1,0
  4541.0    0.05       0  4900.0    0.12       0  5016.1    0.07       0
  5022.4    0.12       0  5262.5    0.05       0
Bank Sta=5016.1,5022.4
Exp/Cntr=0.3,0.1

Type RM Length L Ch R = 1,49841,961,961,961
BEGIN DESCRIPTION:
MILLER CREEK 89.0
END DESCRIPTION:
XS GIS Cut Line= 3
      2866005.67     10277503.07      2865881.50     10277116.00
      2865705.67     10276953.09
#Sta/Elev= 30
  4593.5 1165.30  4641.6 1163.37  4646.9 1164.09  4668.5 1163.39  4698.5 1163.05
  4719.5 1164.13  4775.4 1163.57  4814.0 1161.28  4834.4 1158.97  4839.6 1159.66
  4866.5 1157.12  4877.0 1154.52  4898.0 1151.38  4903.9 1152.21  4909.1 1150.84
  4968.1 1151.97  4995.7 1149.38  4996.2 1148.88  5002.0 1149.38  5006.4 1152.65
  5020.5 1158.68  5055.7 1162.09  5069.9 1162.72  5076.7 1162.14  5105.0 1164.10
  5126.6 1163.32  5183.3 1163.97  5197.4 1164.89  5232.6 1164.72  5239.7 1165.56
#Mann=4,-1,0
  4593.5    0.05       0  4668.5    0.12       0  4995.7    0.07       0
  5002.0    0.12       0
Bank Sta=4995.7,5002
Exp/Cntr=0.3,0.1

Type RM Length L Ch R = 1,48880,495,495,495
BEGIN DESCRIPTION:
MILLER CREEK 88.0
END DESCRIPTION:
XS GIS Cut Line= 3
      2866505.67     10277203.09      2866442.50     10277132.00
      2866305.70     10276853.15
#Sta/Elev= 30
  4904.9 1158.79  4926.2 1157.57  4932.9 1156.02  4940.4 1156.66  4947.1 1153.39
  4954.6 1154.75  4961.3 1151.26  4968.8 1150.43  4975.5 1148.10  4983.1 1147.34
  4992.7 1145.12  4993.2 1144.62  4998.6 1144.62  4999.1 1145.12  5002.1 1145.12
  5004.2 1146.32  5009.9 1148.36  5021.0 1149.37  5026.7 1151.05  5032.3 1151.69
  5043.3 1151.67  5049.2 1151.16  5077.3 1153.44  5094.2 1153.44  5099.8 1153.78
  5116.7 1153.50  5132.4 1154.36  5139.2 1153.67  5279.7 1158.15  5310.6 1158.44
#Mann=3,-1,0
  4904.9    0.12       0  4992.7    0.07       0  4999.1    0.12       0
Bank Sta=4992.7,4999.1
Exp/Cntr=0.3,0.1

Type RM Length L Ch R = 1,48385,474,474,474
BEGIN DESCRIPTION:
MILLER CREEK 87.0
END DESCRIPTION:
XS GIS Cut Line= 3
      2866655.73     10276703.12      2866465.75     10276679.00
      2866305.68     10276753.12
#Sta/Elev= 30
  4808.5 1156.94  4838.8 1155.49  4846.0 1154.80  4849.7 1155.25  4851.1 1155.42
  4869.0 1153.03  4926.1 1148.63  4939.6 1148.35  4949.7 1149.17  4969.8 1148.34
  4979.9 1147.51  4990.0 1143.96  4997.5 1142.05  5006.8 1141.81  5007.3 1141.31
  5014.8 1141.31  5015.3 1141.81  5019.1 1144.41  5024.7 1142.72  5033.1 1145.79
  5042.1 1148.24  5047.6 1148.83  5055.2 1150.82  5077.2 1153.19  5106.1 1153.94
  5110.3 1154.04  5116.3 1154.79  5121.8 1154.67  5132.3 1155.78  5176.4 1157.13
#Mann=5,-1,0
  4808.5    0.05       0  4849.7    0.12       0  5006.8    0.07       0
  5015.3    0.12       0  5106.1    0.05       0
Bank Sta=5006.8,5015.3
Exp/Cntr=0.3,0.1

Type RM Length L Ch R = 1,47911,488,488,488
BEGIN DESCRIPTION:
MILLER CREEK 86.0
END DESCRIPTION:
XS GIS Cut Line= 3
      2867005.73     10276203.11      2866628.25     10276245.00
      2865805.71     10276403.11
#Sta/Elev= 30
  4620.2 1160.08  4802.1 1152.46  4821.5 1151.48  4841.6 1151.59  4846.8 1149.94
  4881.8 1144.86  4891.9 1146.68  4912.0 1148.11  4932.2 1148.21  4942.4 1150.17
  4962.3 1151.69  4994.5 1140.68  4995.0 1140.18  5002.5 1140.18  5003.0 1140.68
  5017.2 1141.30  5023.0 1144.37  5069.1 1147.04  5135.0 1148.87  5216.5 1148.67
  5348.8 1151.07  5369.2 1150.06  5420.1 1149.14  5497.8 1151.75  5541.7 1152.77
  5598.8 1155.27  5628.9 1155.62  5695.1 1157.80  5725.6 1157.96  5837.6 1162.57
#Mann=6,-1,0
  4620.2    0.05       0  4802.1    0.12       0  4994.5    0.07       0
  5003.0    0.12       0  5497.8    0.05       0  5628.9    0.12       0
Bank Sta=4994.5,5003
Exp/Cntr=0.3,0.1

Type RM Length L Ch R = 1,47423,444,444,444
BEGIN DESCRIPTION:
MILLER CREEK 85.0
END DESCRIPTION:
XS GIS Cut Line= 3
      2866505.69     10275753.11      2866390.75     10275837.00
      2866105.66     10276103.13
#Sta/Elev= 30
  4857.7 1150.15  4871.2 1149.39  4915.2 1145.20  4944.4 1143.13  4950.8 1141.45
  4957.0 1140.84  4965.5 1141.24  4971.6 1140.88  4995.7 1138.41  4996.2 1137.91
  5003.9 1137.91  5004.4 1138.41  5007.7 1141.68  5015.0 1144.39  5029.2 1145.30
  5050.2 1145.79  5116.0 1144.12  5234.4 1142.31  5255.4 1143.00  5291.0 1142.69
  5297.9 1143.19  5305.2 1142.65  5333.5 1144.25  5340.4 1145.62  5354.6 1147.37
  5361.9 1147.50  5368.7 1149.03  5376.0 1149.10  5382.9 1150.15  5390.0 1150.23
#Mann=4,-1,0
  4857.7    0.05       0  4995.7    0.05       0  5004.4    0.05       0
  5116.0    0.12       0
Bank Sta=4995.7,5004.4
Exp/Cntr=0.3,0.1

Type RM Length L Ch R = 1,46979,480,480,480
BEGIN DESCRIPTION:
MILLER CREEK 84.0
END DESCRIPTION:
XS GIS Cut Line= 3
      2866705.65     10275803.08      2866265.75     10275466.00
      2865855.67     10275753.12
#Sta/Elev= 30
  4445.8 1152.63  4731.3 1150.63  4737.6 1149.22  4802.0 1148.01  4851.9 1143.32
  4916.3 1144.39  4938.0 1143.42  4966.1 1142.12  4980.6 1137.55  4993.9 1136.58
  4994.4 1136.08  5002.6 1136.58  5048.9 1136.91  5055.5 1140.48  5061.6 1139.35
  5070.3 1141.87  5076.4 1141.09  5085.1 1143.00  5091.2 1142.18  5106.1 1144.61
  5141.8 1146.24  5147.9 1145.57  5156.6 1146.69  5162.7 1145.87  5234.2 1147.69
  5263.9 1149.84  5284.8 1149.18  5293.1 1151.02  5320.5 1150.65  5500.6 1155.01
#Mann=4,-1,0
  4445.8    0.12       0  4938.0    0.05       0  4993.9    0.05       0
  5002.6    0.05       0
Bank Sta=4993.9,5002.6
Exp/Cntr=0.3,0.1

Type RM Length L Ch R = 1,46499,491,491,491
BEGIN DESCRIPTION:
MILLER CREEK 83.0
END DESCRIPTION:
XS GIS Cut Line= 3
      2866855.72     10275203.12      2866512.75     10275123.00
      2865505.66     10275003.11
#Sta/Elev= 30
  4647.8 1151.41  4714.2 1149.23  4755.2 1146.71  4822.4 1143.45  4841.7 1141.75
  4846.9 1142.24  4853.2 1140.37  4863.5 1142.63  4884.0 1144.24  4894.5 1143.96
  4931.9 1145.98  4955.9 1146.35  4966.2 1142.21  4974.4 1137.76  4979.6 1138.10
  4986.7 1136.60  5000.0 1136.46  5012.8 1134.86  5013.3 1134.36  5021.6 1134.86
  5027.3 1139.26  5047.4 1141.82  5067.5 1140.35  5126.2 1141.49  5212.1 1145.71
  5289.1 1146.63  5722.6 1146.95  5805.2 1149.79  5843.0 1151.83  6014.2 1154.96
#Mann=5,-1,0
  4647.8    0.05       0  4755.2    0.12       0  5012.8    0.07       0
  5021.6    0.12       0  5126.2    0.05       0
Bank Sta=5012.8,5021.6
Exp/Cntr=0.3,0.1

Type RM Length L Ch R = 1,46008,480,480,480
BEGIN DESCRIPTION:
MILLER CREEK 82.0
END DESCRIPTION:
XS GIS Cut Line= 3
      2867005.66     10275253.09      2866537.75     10274657.00
      2865555.66     10274653.11
#Sta/Elev= 30
  4242.2 1155.31  4455.7 1151.12  4490.3 1150.38  4671.6 1143.23  4798.0 1140.13
  4876.7 1141.01  4883.0 1139.95  4890.5 1142.26  4898.4 1141.43  4925.7 1140.25
  4940.8 1139.79  4947.2 1138.25  4961.7 1139.38  4968.0 1136.68  4976.1 1136.60
  4982.5 1134.60  4990.6 1135.37  4992.5 1133.01  4993.0 1132.51  5001.3 1133.01
  5008.8 1133.35  5032.1 1138.09  5062.1 1137.50  5092.1 1140.20  5139.3 1142.18
  5444.3 1144.89  5534.4 1145.22  5642.1 1145.48  5772.1 1149.90  5982.1 1153.82
#Mann=12,-1,0
  4242.2    0.12       0  4455.7    0.05       0  4490.3    0.12       0
  4671.6    0.05       0  4898.4    0.12       0  4925.7    0.05       0
  4992.5    0.05       0  5001.3    0.05       0  5008.8    0.12       0
  5139.3    0.05       0  5444.3    0.12       0  5534.4    0.05       0
Bank Sta=4992.5,5001.3
Exp/Cntr=0.3,0.1

Type RM Length L Ch R = 1,45528,1365,1365,1365
BEGIN DESCRIPTION:
MILLER CREEK 81.0
END DESCRIPTION:
XS GIS Cut Line= 3
      2866955.69     10274753.12      2866669.00     10274260.00
      2865955.71     10274403.11
#Sta/Elev= 30
  4429.6 1147.61  4502.0 1145.60  4544.2 1143.57  4576.5 1143.30  4619.5 1140.99
  4656.8 1141.14  4662.6 1140.17  4721.3 1138.59  4810.8 1137.75  4891.8 1136.35
  4972.1 1136.66  4984.8 1133.34  5009.0 1132.24  5009.5 1131.74  5017.6 1131.74
  5018.1 1132.24  5023.8 1132.94  5040.2 1136.65  5045.3 1135.15  5064.6 1138.43
  5074.8 1139.34  5142.0 1140.52  5153.5 1140.18  5192.9 1141.20  5309.4 1141.92
  5329.8 1142.78  5482.7 1142.96  5564.3 1144.44  5600.2 1146.31  5727.5 1147.89
#Mann=6,-1,0
  4429.6    0.05       0  4544.2    0.12       0  4810.8    0.05       0
  5009.0    0.05       0  5018.1    0.05       0  5153.5    0.12       0
Bank Sta=5009,5018.1
Exp/Cntr=0.3,0.1

Type RM Length L Ch R = 1,44163,478,478,478
BEGIN DESCRIPTION:
MILLER CREEK 80.0
END DESCRIPTION:
XS GIS Cut Line= 3
      2867555.65     10273603.10      2867150.25     10273429.00
      2865955.67     10274353.12
#Sta/Elev= 30
  4558.8 1142.41  4580.5 1142.55  4634.5 1139.21  4656.7 1137.77  4672.9 1138.38
  4678.5 1137.23  4720.0 1134.70  4749.0 1134.47  4772.6 1133.26  4917.9 1131.64
  4948.3 1128.75  4953.8 1129.06  4971.9 1127.63  4977.3 1128.26  4989.3 1127.20
  4989.8 1126.70  4998.9 1127.20  4999.8 1127.95  5006.0 1127.95  5028.0 1132.65
  5060.2 1133.66  5156.6 1134.19  5292.0 1136.70  5519.7 1138.66  6181.6 1141.81
  6223.1 1142.62  6368.1 1144.81  6492.0 1148.28  6497.3 1148.41  6510.3 1148.04
#Mann=9,-1,0
  4558.8    0.12       0  4634.5    0.05       0  4989.3    0.05       0
  4998.9    0.05       0  5060.2    0.12       0  5292.0    0.05       0
  6223.1    0.12       0  6492.0    0.05       0  6497.3    0.12       0
Bank Sta=4989.3,4998.9
Exp/Cntr=0.3,0.1

Type RM Length L Ch R = 1,43685,1790,1790,1790
BEGIN DESCRIPTION:
MILLER CREEK 79.0
END DESCRIPTION:
XS GIS Cut Line= 3
      2867455.68     10273153.11      2867234.75     10273044.00
      2866155.65     10273353.12
#Sta/Elev= 30
  4753.6 1140.44  4784.8 1139.13  4866.8 1135.89  4879.8 1136.12  4896.7 1133.42
  4902.3 1134.79  4919.1 1127.04  4924.7 1130.45  4941.6 1126.34  4947.2 1128.88
  4954.3 1125.94  4964.0 1125.21  4969.6 1126.47  4991.9 1124.98  4992.4 1124.48
  5001.5 1124.98  5048.5 1130.85  5061.4 1131.26  5121.3 1130.23  5199.2 1131.67
  5238.3 1129.94  5339.4 1129.58  5344.6 1130.51  5451.1 1130.86  5559.4 1134.38
  5591.3 1135.61  5807.8 1136.17  5976.8 1139.95  6102.7 1140.80  6122.5 1141.08
#Mann=8,-1,0
  4753.6    0.12       0  4784.8    0.05       0  4866.8    0.12       0
  4991.9    0.07       0  5001.5    0.12       0  5559.4    0.05       0
  5807.8    0.12       0  6102.7    0.05       0
Bank Sta=4991.9,5001.5
Exp/Cntr=0.3,0.1

Type RM Length L Ch R = 1,41895,766,766,766
BEGIN DESCRIPTION:
Mapping XS 2cdccd61
END DESCRIPTION:
XS GIS Cut Line= 3
      2867940.31     10272122.23      2866565.31     10272122.23
      2865670.05     10272143.05
#Sta/Elev= 30
  3782.8 1146.34  3817.4 1146.71  4147.4 1140.94  4327.4 1136.04  4527.4 1127.87
  4757.4 1122.96  4867.4 1122.96  4907.4 1121.73  4937.4 1123.31  4967.4 1123.13
  4977.4 1121.64  4982.5 1119.71  4983.0 1119.21  4992.4 1119.71  5007.4 1119.92
  5027.4 1123.55  5057.4 1124.77  5117.4 1125.24  5215.8 1124.04  5257.5 1123.69
  5337.5 1125.97  5417.5 1123.62  5457.5 1120.80  5477.5 1122.33  5611.4 1125.80
  5797.6 1132.43  5807.6 1131.67  5887.6 1134.77  5947.8 1135.70  6053.3 1136.81
#Mann=6,-1,0
  3782.8    0.05       0  4982.5    0.03       0  4992.4    0.05       0
  5215.8    0.12       0  5611.4    0.05       0  5947.8    0.12       0
Bank Sta=4982.5,4992.4
Exp/Cntr=0.3,0.1

Type RM Length L Ch R = 1,41129,212,212,212
BEGIN DESCRIPTION:
Mapping XS 3c1f6463
END DESCRIPTION:
XS GIS Cut Line= 4
      2868190.33     10271663.89      2866836.14     10271663.89
      2866315.31     10271705.56      2865920.03     10271830.38
#Sta/Elev= 30
  2984.9 1141.63  3329.5 1147.26  3422.1 1146.97  3909.5 1136.07  3989.5 1136.34
  4019.5 1137.98  4069.5 1143.16  4109.5 1140.16  4139.5 1136.09  4189.5 1135.68
  4229.5 1132.64  4253.1 1132.45  4375.9 1129.00  4425.0 1128.17  4550.2 1126.68
  4720.8 1121.83  4821.1 1122.74  4892.7 1120.97  4913.6 1121.81  4973.9 1117.11
  5002.9 1114.58  5003.4 1114.08  5013.3 1114.58  5029.0 1117.50  5035.2 1121.27
  5050.0 1123.93  5105.1 1124.95  5169.7 1128.23  5196.8 1130.94  5276.1 1130.86
#Mann=8,-1,0
  2984.9    0.12       0  3422.1    0.05       0  4253.1    0.12       0
  4375.9    0.05       0  4425.0    0.12       0  4973.9    0.05       0
  5002.9    0.05       0  5013.3    0.05       0
Bank Sta=5002.9,5013.3
Exp/Cntr=0.3,0.1

Type RM Length L Ch R = 1,40917,474,474,474
BEGIN DESCRIPTION:
MILLER CREEK 74.0
END DESCRIPTION:
XS GIS Cut Line= 3
      2866855.68     10271503.11      2866144.00     10271554.00
      2866055.64     10271603.13
#Sta/Elev= 30
  4286.5 1135.97  4316.6 1133.35  4396.8 1130.41  4406.8 1129.39  4446.9 1129.43
  4467.0 1127.88  4494.4 1127.23  4499.4 1127.62  4517.1 1126.59  4610.0 1124.47
  4657.4 1123.79  4687.5 1122.51  4697.5 1123.14  4747.7 1120.53  4775.0 1119.80
  4880.8 1121.28  4908.1 1120.38  4938.2 1120.54  4964.1 1119.17  4978.3 1117.46
  4988.3 1114.24  5000.9 1114.20  5001.4 1113.70  5010.8 1113.70  5011.3 1114.20
  5021.0 1115.41  5033.6 1120.12  5043.8 1125.03  5049.6 1126.56  5101.1 1129.70
#Mann=6,-1,0
  4286.5    0.05       0  4610.0    0.12       0  4880.8    0.05       0
  4964.1    0.12       0  5000.9    0.07       0  5011.3    0.12       0
Bank Sta=5000.9,5011.3
Exp/Cntr=0.3,0.1

Type RM Length L Ch R = 1,40443,469,469,469
BEGIN DESCRIPTION:
MILLER CREEK 73.0
END DESCRIPTION:
XS GIS Cut Line= 3
      2866655.67     10270753.13      2866319.00     10271116.00
      2865905.65     10271403.14
#Sta/Elev= 30
  4505.0 1135.72  4709.9 1123.77  4724.1 1123.32  4731.5 1126.24  4752.5 1125.00
  4759.8 1126.75  4766.6 1124.08  4788.2 1124.10  4795.0 1122.08  4802.3 1123.46
  4809.1 1120.54  4816.5 1121.29  4837.5 1117.89  4870.0 1118.87  4929.3 1120.25
  4950.9 1117.98  4957.7 1114.02  4965.0 1115.49  4971.9 1112.02  4979.2 1113.65
  5001.7 1111.85  5002.2 1111.35  5012.1 1111.85  5021.8 1112.47  5036.6 1116.95
  5042.7 1115.29  5072.4 1118.77  5101.3 1119.05  5245.3 1119.79  5503.3 1130.59
#Mann=5,-1,0
  4505.0    0.05       0  4870.0    0.12       0  5001.7    0.07       0
  5012.1    0.12       0  5101.3    0.05       0
Bank Sta=5001.7,5012.1
Exp/Cntr=0.3,0.1

Type RM Length L Ch R = 1,39974,481,481,481
BEGIN DESCRIPTION:
MILLER CREEK 72.0
END DESCRIPTION:
XS GIS Cut Line= 3
      2866305.70     10270703.11      2866119.00     10270726.00
      2865905.67     10270953.12
#Sta/Elev= 30
  4811.9 1127.36  4822.0 1127.55  4832.1 1125.84  4846.0 1124.32  4855.1 1123.17
  4862.3 1120.09  4872.4 1118.80  4912.7 1116.85  4931.5 1116.65  4973.1 1114.06
  4993.9 1109.69  4994.4 1109.19  5003.9 1109.19  5004.4 1109.69  5014.4 1115.11
  5028.5 1115.48  5042.7 1114.87  5085.2 1116.71  5092.1 1116.07  5120.4 1115.55
  5141.8 1115.90  5156.0 1115.47  5170.4 1115.94  5177.0 1116.44  5184.3 1116.13
  5191.2 1117.49  5212.7 1118.15  5219.5 1118.99  5290.3 1124.12  5311.6 1124.64
#Mann=5,-1,0
  4811.9    0.05       0  4846.0    0.12       0  4993.9    0.07       0
  5004.4    0.12       0  5170.4    0.05       0
Bank Sta=4993.9,5004.4
Exp/Cntr=0.3,0.1

Type RM Length L Ch R = 1,39493,475,475,475
BEGIN DESCRIPTION:
MILLER CREEK 71.0
END DESCRIPTION:
XS GIS Cut Line= 3
      2866155.69     10270103.11      2865737.75     10270466.00
      2865805.68     10271203.08
#Sta/Elev= 30
  4446.5 1131.71  4449.8 1131.71  4453.6 1129.71  4460.3 1129.57  4467.9 1128.22
  4474.5 1127.95  4496.4 1123.50  4503.0 1124.29  4510.6 1121.69  4737.6 1114.46
  4822.1 1114.11  4843.8 1113.21  4899.9 1114.40  4971.2 1113.88  4985.4 1113.08
  4992.0 1110.21  4998.1 1109.62  5026.8 1108.95  5027.3 1108.45  5036.9 1108.45
  5037.4 1108.95  5047.3 1113.64  5057.4 1114.31  5141.8 1116.52  5212.4 1119.45
  5278.3 1121.65  5356.2 1121.83  5509.5 1124.43  5659.9 1126.99  5740.2 1129.31
#Mann=5,-1,0
  4446.5    0.05       0  5026.8    0.05       0  5037.4    0.05       0
  5212.4    0.12       0  5509.5    0.05       0
Bank Sta=5026.8,5037.4
Exp/Cntr=0.3,0.1

Type RM Length L Ch R = 1,39018,440,440,440
BEGIN DESCRIPTION:
MILLER CREEK 70.0
END DESCRIPTION:
XS GIS Cut Line= 3
      2865905.66     10269803.13      2865503.25     10270135.00
      2865205.69     10271353.08
#Sta/Elev= 30
  4478.4 1127.92  4549.4 1125.04  4578.1 1123.11  4606.7 1122.99  4634.0 1121.85
  4766.9 1115.36  4841.3 1111.36  4913.7 1111.44  4954.6 1112.52  4968.9 1111.29
  4975.4 1107.51  4989.8 1107.47  4990.3 1106.97  5000.5 1107.47  5012.2 1108.13
  5018.6 1110.97  5028.9 1112.22  5053.8 1110.54  5080.4 1112.43  5090.3 1112.51
  5095.5 1111.72  5152.5 1111.94  5225.6 1113.39  5308.9 1113.67  5388.4 1115.32
  5395.2 1115.15  5541.7 1117.11  5718.6 1121.19  5923.7 1123.66  6253.9 1127.53
#Mann=9,-1,0
  4478.4    0.05       0  4766.9    0.12       0  4913.7    0.05       0
  4989.8    0.05       0  5000.5    0.05       0  5388.4    0.12       0
  5395.2    0.05       0  5541.7    0.12       0  5923.7    0.05       0
Bank Sta=4989.8,5000.5
Exp/Cntr=0.3,0.1

Type RM Length L Ch R = 1,38578,484,484,484
BEGIN DESCRIPTION:
MILLER CREEK 69.0
END DESCRIPTION:
XS GIS Cut Line= 3
      2865655.65     10269453.14      2865340.75     10269748.00
      2864805.66     10270003.12
#Sta/Elev= 30
  4568.6 1132.56  4572.0 1132.56  4575.6 1130.93  4582.5 1130.42  4596.7 1126.64
  4618.1 1122.78  4632.3 1120.77  4639.1 1121.17  4674.8 1117.48  4731.5 1114.65
  4780.8 1115.29  4901.2 1110.47  4915.1 1108.77  4964.9 1109.44  4986.0 1105.07
  5000.0 1104.17  5000.4 1103.09  5000.9 1102.59  5011.1 1103.09  5016.7 1109.01
  5022.9 1110.13  5083.1 1109.20  5120.0 1109.30  5230.4 1109.80  5255.4 1108.84
  5315.8 1110.46  5374.4 1109.94  5419.8 1111.15  5436.9 1112.58  5592.8 1115.59
#Mann=7,-1,0
  4568.6    0.05       0  4901.2    0.12       0  5000.4    0.07       0
  5011.1    0.12       0  5083.1    0.05       0  5120.0    0.12       0
  5230.4    0.05       0
Bank Sta=5000.4,5011.1
Exp/Cntr=0.3,0.1

Type RM Length L Ch R = 1,38094,494,494,494
BEGIN DESCRIPTION:
MILLER CREEK 68.0
END DESCRIPTION:
XS GIS Cut Line= 3
      2865505.73     10269303.11      2865128.25     10269323.00
      2863905.69     10270203.11
#Sta/Elev= 30
  4622.0 1122.00  4652.1 1118.69  4662.1 1119.50  4702.2 1115.66  4732.2 1115.81
  4832.3 1110.90  4891.0 1106.76  4912.4 1106.16  4962.5 1107.93  4972.5 1106.75
  4993.4 1101.73  4993.9 1101.23  5004.2 1101.73  5009.0 1102.21  5015.5 1107.34
  5023.8 1108.10  5059.4 1106.30  5088.8 1106.86  5145.3 1105.21  5174.7 1106.43
  5185.0 1105.07  5281.5 1109.03  5459.9 1112.63  5670.9 1115.97  5847.3 1116.83
  6013.0 1115.78  6107.7 1117.68  6376.9 1123.33  6461.6 1125.41  6506.4 1126.01
#Mann=10,-1,0
  4622.0    0.05       0  4891.0    0.12       0  4993.4    0.07       0
  5004.2    0.12       0  5185.0    0.05       0  5459.9    0.12       0
  5670.9    0.05       0  6107.7    0.12       0  6376.9    0.05       0
  6461.6    0.12       0
Bank Sta=4993.4,5004.2
Exp/Cntr=0.3,0.1
