--- REED CREEK.prj (project) ---

Proj Title=REED CREEK Base Level Engineering
Current Plan=p01
Default Exp/Contr=0.3,0.1
English Units
Geom File=g01
Flow File=f01
Plan File=p01
Y Axis Title=Elevation
X Axis Title(PF)=Main Channel Distance
X Axis Title(XS)=Station
BEGIN DESCRIPTION:
REED CREEK
END DESCRIPTION:
DSS Export Rating Curves= 0
DSS Export Rating Curve Sorted= 0
DSS Export Volume Flow Curves= 0
DXF OffsetX= 0
DXF OffsetY= 0
DXF ScaleX= 1
DXF ScaleY= 10

--- REED CREEK.p01 (plan) ---

Plan Title=Multiple Run
Short Identifier=Multiple
Geom File=g01
Flow File=f01
Subcritical Flow
K Sum by GR= 0
Std Step Tol= 0.01
Critical Tol= 0.01
Num of Std Step Trials= 20
Max Error Tol= 0.3
Flow Tol Ratio= 0.001
Split Flow NTrial= 30
Split Flow Tol= 0.02
Split Flow Ratio= 0.02
Log Output Level= 0
Friction Slope Method= 1
Unsteady Friction Slope Method= 2
Unsteady Bridges Friction Slope Method= 1
Parabolic Critical Depth
Global Vel Dist=  1 , 1 , 1
Global Log Level= 0
CheckData=True
Encroach Param= -1, 0, 0, 0
BEGIN DESCRIPTION:
Multiple Run
END DESCRIPTION:

--- REED CREEK.f01 (steady flow) ---

Flow Title=Multiple
Program Version=4.10
Number of Profiles= 7
Profile Names=10-year,25-year,50-year,1pct_min,100-year,1pct_plu,500-year
River Rch & RM=REED CREEK,Reach-1         ,32933
      67     127     197     102     307     927     805
River Rch & RM=REED CREEK,Reach-1         ,23173
      94     186     296     156     471    1423    1277
River Rch & RM=REED CREEK,Reach-1         ,16772
     131     273     443     237     716    2162    1996
River Rch & RM=REED CREEK,Reach-1         ,12092
     134     280     455     244     736    2223    2056
River Rch & RM=REED CREEK,Reach-1         ,11098
     220     483     804     439    1327    4006    3838
River Rch & RM=REED CREEK,Reach-1         ,4410
     222     490     816     446    1348    4071    3904
River Rch & RM=REED CREEK,Reach-1         ,3464
     329     744    1258     696    2103    6351    6232
Boundary for River Rch & Prof#=REED CREEK,Reach-1         , 1
Up Type= 0
Dn Type= 3
Dn Slope=0.0005
Boundary for River Rch & Prof#=REED CREEK,Reach-1         , 2
Up Type= 0
Dn Type= 3
Dn Slope=0.0005
Boundary for River Rch & Prof#=REED CREEK,Reach-1         , 3
Up Type= 0
Dn Type= 3
Dn Slope=0.0005
Boundary for River Rch & Prof#=REED CREEK,Reach-1         , 4
Up Type= 0
Dn Type= 3
Dn Slope=0.0005
Boundary for River Rch & Prof#=REED CREEK,Reach-1         , 5
Up Type= 0
Dn Type= 3
Dn Slope=0.0005
Boundary for River Rch & Prof#=REED CREEK,Reach-1         , 6
Up Type= 0
Dn Type= 3
Dn Slope=0.0005
Boundary for River Rch & Prof#=REED CREEK,Reach-1         , 7
Up Type= 0
Dn Type= 3
Dn Slope=0.0005
DSS Import GetInterval= 0
DSS Import GetPeak= 0
DSS Import FillOption= 0

--- REED CREEK.g01 (geometry) ---

Geom Title=Existing Conditions

River Reach=REED CREEK,Reach-1
Reach XY= 30
      2827157.00     10276735.00      2827671.75     10275767.00
      2828390.50     10275590.00      2828668.75     10275048.00
      2828807.75     10272605.00      2829452.50     10271441.00
      2829331.50     10270601.00      2828755.00     10270142.00
      2829366.25     10270076.00      2829671.75     10269695.00
      2830407.25     10269993.00      2833735.00     10268794.00
      2834171.25     10269041.00      2835102.25     10268781.00
      2835932.25     10269198.00      2836598.75     10268287.00
      2837317.75     10267946.00      2837967.50     10268487.00
      2838376.25     10268533.00      2838710.00     10267514.00
      2839460.00     10267403.00      2839939.00     10267719.00
      2841601.50     10267368.00      2842233.50     10266625.00
      2842454.25     10265395.00      2844115.50     10263993.00
      2844271.75     10262545.00      2845178.00     10262392.00
      2845969.50     10262944.00      2847424.75     10262690.00

Type RM Length L Ch R = 1,32933,432,432,432
BEGIN DESCRIPTION:
REED CREEK 68.0
END DESCRIPTION:
XS GIS Cut Line= 3
      2827655.67     10276653.09      2827382.50     10276370.00
      2827255.70     10276453.10
#Sta/Elev= 30
  4606.6 1397.10  4613.7 1397.68  4620.6 1395.94  4627.8 1390.43  4634.7 1389.69
  4656.1 1383.29  4679.4 1383.27  4698.5 1380.98  4712.7 1380.72  4726.8 1375.96
  4741.0 1370.30  4769.3 1366.00  4896.6 1356.27  4939.1 1354.40  4946.0 1355.04
  4953.2 1354.23  4960.2 1354.72  4967.4 1353.83  4988.5 1346.92  4992.4 1346.80
  4992.6 1343.80  4996.1 1343.80  4996.4 1346.80  5008.1 1347.83  5020.4 1351.69
  5029.6 1353.43  5086.8 1359.28  5115.8 1360.65  5129.0 1362.65  5151.6 1364.23
#Mann=4,-1,0
  4606.6    0.12       0  4679.4    0.05       0  4992.4    0.05       0
  4996.4    0.05       0
Bank Sta=4992.4,4996.4
Exp/Cntr=0.3,0.1

Type RM Length L Ch R = 1,32501,410,410,410
BEGIN DESCRIPTION:
REED CREEK 67.0
END DESCRIPTION:
XS GIS Cut Line= 3
      2827855.71     10276253.14      2827532.25     10275968.00
      2827255.65     10275953.11
#Sta/Elev= 30
  4568.8 1366.48  4611.1 1359.84  4647.1 1355.84  4653.8 1356.05  4661.3 1354.15
  4675.5 1353.43  4688.9 1350.32  4710.3 1347.96  4759.4 1342.35  4781.8 1343.27
  4788.5 1342.75  4802.7 1343.95  4894.7 1338.95  4908.9 1339.04  4929.8 1337.10
  4951.6 1337.13  4986.7 1333.57  5004.6 1329.62  5004.8 1326.62  5008.3 1326.62
  5008.6 1329.62  5016.6 1333.58  5036.6 1337.33  5066.7 1339.64  5116.7 1340.63
  5136.8 1343.76  5176.8 1346.15  5182.9 1346.75  5187.9 1348.49  5277.0 1357.24
#Mann=5,-1,0
  4568.8    0.05       0  4710.3    0.12       0  4759.4    0.05       0
  5004.6    0.05       0  5008.6    0.05       0
Bank Sta=5004.6,5008.6
Exp/Cntr=0.3,0.1

Type RM Length L Ch R = 1,32091,474,474,474
BEGIN DESCRIPTION:
REED CREEK 66.0
END DESCRIPTION:
XS GIS Cut Line= 3
      2827855.67     10275753.10      2827814.00     10275695.00
      2827755.68     10275653.11
#Sta/Elev= 27
  4928.5 1326.57  4931.6 1326.57  4935.8 1325.18  4942.0 1325.20  4950.6 1324.08
  4956.7 1324.04  4965.3 1322.45  4971.5 1322.37  4977.7 1319.24  4984.2 1316.57
  4984.4 1313.57  4987.9 1313.57  4988.2 1316.57  4992.4 1316.77  4998.1 1317.74
  5002.0 1317.74  5007.9 1317.79  5014.1 1319.47  5022.6 1320.00  5028.8 1320.15
  5035.0 1321.51  5043.6 1322.41  5049.7 1324.37  5058.3 1326.03  5064.4 1326.42
  5068.7 1326.89  5071.8 1326.89
#Mann=3,-1,0
  4928.5    0.05       0  4984.2    0.05       0  4988.2    0.05       0
Bank Sta=4984.2,4988.2
Exp/Cntr=0.3,0.1

Type RM Length L Ch R = 1,31617,470,470,470
BEGIN DESCRIPTION:
REED CREEK 65.0
END DESCRIPTION:
XS GIS Cut Line= 3
      2828155.69     10275903.08      2828261.25     10275590.00
      2828205.70     10275503.14
#Sta/Elev= 30
  4669.6 1342.75  4711.5 1340.19  4722.3 1337.31  4743.0 1335.18  4748.3 1332.71
  4774.5 1329.93  4779.8 1328.03  4785.7 1327.21  4806.0 1326.16  4811.2 1324.05
  4827.5 1322.25  4922.8 1315.53  4937.2 1313.67  4944.0 1311.91  4968.6 1309.24
  4975.6 1306.72  4986.2 1304.48  4997.1 1303.33  4997.4 1300.33  5000.9 1300.33
  5001.1 1303.33  5008.2 1304.73  5016.9 1308.18  5022.8 1307.22  5038.0 1311.91
  5074.4 1314.97  5080.3 1314.80  5089.6 1316.06  5095.5 1315.81  5103.1 1316.83
#Mann=4,-1,0
  4669.6    0.12       0  4827.5    0.05       0  4997.1    0.05       0
  5001.1    0.05       0
Bank Sta=4997.1,5001.1
Exp/Cntr=0.3,0.1

Type RM Length L Ch R = 1,31147,484,484,484
BEGIN DESCRIPTION:
REED CREEK 64.0
END DESCRIPTION:
XS GIS Cut Line= 3
      2828555.71     10275353.15      2828497.25     10275274.00
      2828455.67     10275203.09
#Sta/Elev= 30
  4901.6 1302.73  4904.8 1302.73  4909.0 1302.28  4915.2 1302.45  4923.6 1302.25
  4938.2 1300.83  4944.4 1300.15  4951.4 1299.27  4959.1 1298.58  4965.3 1298.16
  4973.7 1297.26  4980.1 1296.85  4988.3 1295.08  4994.6 1293.13  4995.4 1291.81
  4995.7 1288.81  4999.2 1288.81  4999.4 1291.81  5003.4 1291.81  5009.9 1292.23
  5015.7 1297.08  5024.2 1300.94  5031.4 1304.00  5037.2 1305.25  5047.1 1306.02
  5052.9 1307.89  5059.0 1309.54  5068.5 1310.12  5074.3 1310.96  5082.2 1311.07
#Mann=4,-1,0
  4901.6    0.12       0  4980.1    0.05       0  4995.4    0.05       0
  4999.4    0.05       0
Bank Sta=4995.4,4999.4
Exp/Cntr=0.3,0.1

Type RM Length L Ch R = 1,30663,476,476,476
BEGIN DESCRIPTION:
REED CREEK 63.0
END DESCRIPTION:
XS GIS Cut Line= 3
      2828855.68     10274853.11      2828681.50     10274856.00
      2828505.72     10274853.11
#Sta/Elev= 30
  4825.8 1297.48  4835.8 1297.33  4865.8 1295.17  4875.8 1291.96  4895.8 1288.66
  4905.8 1288.81  4915.8 1289.62  4925.3 1289.41  4935.8 1289.14  4955.8 1288.14
  4965.8 1286.65  4975.8 1286.63  4995.4 1285.82  5000.0 1285.82  5003.8 1285.48
  5004.1 1282.48  5007.6 1282.48  5007.8 1285.48  5015.8 1287.18  5035.8 1293.36
  5045.8 1294.56  5065.8 1297.38  5075.8 1299.49  5085.8 1301.89  5095.8 1304.42
  5135.8 1315.59  5155.8 1320.90  5165.8 1323.88  5173.3 1326.41  5175.8 1326.41
#Mann=4,-1,0
  4825.8    0.12       0  4925.3    0.05       0  5003.8    0.05       0
  5007.8    0.05       0
Bank Sta=5003.8,5007.8
Exp/Cntr=0.3,0.1

Type RM Length L Ch R = 1,30187,468,468,468
BEGIN DESCRIPTION:
REED CREEK 62.0
END DESCRIPTION:
XS GIS Cut Line= 3
      2828805.67     10274453.10      2828714.75     10274391.00
      2828405.64     10274603.14
#Sta/Elev= 30
  4889.9 1290.98  4927.7 1288.64  4933.2 1288.51  4939.3 1287.13  4948.2 1288.01
  4962.5 1284.60  4969.1 1281.88  4988.1 1278.62  4988.4 1275.62  4991.9 1275.62
  4992.1 1278.62  5014.8 1280.86  5029.7 1284.38  5050.7 1287.32  5059.5 1287.71
  5065.6 1288.79  5071.6 1292.26  5095.4 1292.75  5116.3 1289.90  5180.8 1294.44
  5194.1 1297.40  5209.0 1297.43  5223.9 1299.34  5253.6 1303.71  5302.1 1313.25
  5310.6 1313.86  5338.5 1318.38  5361.3 1323.89  5371.8 1327.73  5374.9 1327.73
#Mann=4,-1,0
  4889.9    0.12       0  4927.7    0.05       0  4988.1    0.05       0
  4992.1    0.05       0
Bank Sta=4988.1,4992.1
Exp/Cntr=0.3,0.1

Type RM Length L Ch R = 1,29719,496,496,496
BEGIN DESCRIPTION:
REED CREEK 61.0
END DESCRIPTION:
XS GIS Cut Line= 3
      2829105.72     10274203.14      2828827.50     10273955.00
      2828705.66     10274003.12
#Sta/Elev= 30
  4627.2 1313.79  4639.6 1312.69  4712.1 1303.48  4733.8 1299.56  4754.7 1296.59
  4761.4 1296.44  4769.0 1294.53  4789.9 1292.80  4825.8 1288.22  4871.4 1283.59
  4889.3 1281.00  4903.6 1279.76  4910.3 1280.00  4938.7 1276.02  4960.4 1274.64
  4988.8 1274.06  4995.5 1272.81  4995.9 1270.49  4996.1 1267.49  4999.6 1267.49
  4999.9 1270.49  5003.7 1270.49  5013.3 1272.49  5032.3 1279.14  5062.0 1281.97
  5086.4 1282.45  5098.7 1283.19  5116.1 1285.71  5121.5 1284.87  5131.0 1286.00
#Mann=5,-1,0
  4627.2    0.12       0  4639.6    0.05       0  4871.4    0.12       0
  4995.9    0.07       0  4999.9    0.12       0
Bank Sta=4995.9,4999.9
Exp/Cntr=0.3,0.1

Type RM Length L Ch R = 1,29223,478,478,478
BEGIN DESCRIPTION:
REED CREEK 60.0
END DESCRIPTION:
XS GIS Cut Line= 3
      2828955.66     10273553.09      2828839.25     10273463.00
      2828555.68     10273253.11
#Sta/Elev= 30
  4852.8 1277.77  4930.6 1273.77  4938.8 1271.60  4945.1 1273.01  4953.3 1269.29
  4959.6 1271.31  4974.1 1262.54  4980.4 1263.69  4992.9 1262.13  4993.2 1259.13
  4996.7 1259.13  4996.9 1262.13  4999.1 1263.07  5038.7 1264.56  5109.6 1263.59
  5124.3 1265.39  5146.8 1266.02  5159.7 1265.07  5174.3 1268.95  5195.2 1269.69
  5209.8 1273.12  5216.0 1272.72  5224.4 1274.71  5230.7 1274.59  5265.9 1281.90
  5295.4 1285.65  5324.6 1292.40  5345.5 1294.92  5349.7 1298.54  5352.8 1298.54
#Mann=5,-1,0
  4852.8    0.12       0  4992.9    0.07       0  4996.9    0.12       0
  5146.8    0.05       0  5265.9    0.12       0
Bank Sta=4992.9,4996.9
Exp/Cntr=0.3,0.1

Type RM Length L Ch R = 1,28745,467,467,467
BEGIN DESCRIPTION:
REED CREEK 59.0
END DESCRIPTION:
XS GIS Cut Line= 3
      2829055.71     10273203.13      2828759.75     10273037.00
      2828455.67     10273153.12
#Sta/Elev= 30
  4660.6 1279.53  4668.6 1280.62  4676.9 1278.32  4696.0 1273.43  4727.9 1270.26
  4733.7 1270.50  4771.3 1266.63  4854.1 1263.04  4955.0 1259.44  4970.3 1258.71
  4992.6 1255.97  5004.4 1255.92  5004.7 1252.92  5008.2 1252.92  5008.4 1255.92
  5015.1 1258.35  5025.8 1259.98  5031.1 1261.49  5061.2 1264.34  5110.6 1276.39
  5116.0 1276.57  5122.1 1278.68  5140.7 1282.21  5176.1 1286.99  5207.7 1292.24
  5218.4 1293.15  5239.8 1297.78  5255.7 1300.06  5310.4 1316.59  5325.5 1317.52
#Mann=5,-1,0
  4660.6    0.12       0  4676.9    0.05       0  4854.1    0.12       0
  5004.4    0.07       0  5008.4    0.12       0
Bank Sta=5004.4,5008.4
Exp/Cntr=0.3,0.1

Type RM Length L Ch R = 1,28278,488,488,488
BEGIN DESCRIPTION:
REED CREEK 58.0
END DESCRIPTION:
XS GIS Cut Line= 3
      2829105.67     10272503.12      2828822.50     10272578.00
      2828505.72     10272453.13
#Sta/Elev= 30
  4707.1 1273.13  4724.6 1270.81  4748.5 1269.56  4758.8 1268.22  4764.9 1266.64
  4805.1 1263.16  4840.2 1253.58  4845.4 1253.85  4851.9 1252.22  4863.2 1252.44
  4885.6 1253.36  4903.6 1252.64  4966.1 1253.55  4986.4 1253.23  5016.1 1250.96
  5016.3 1247.96  5019.8 1247.96  5020.1 1250.96  5079.3 1252.26  5084.7 1256.11
  5103.7 1257.85  5109.1 1260.13  5125.6 1260.38  5133.5 1259.04  5138.9 1260.33
  5147.1 1260.88  5168.6 1264.23  5222.8 1267.25  5301.3 1274.44  5340.5 1281.14
#Mann=4,-1,0
  4707.1    0.12       0  4863.2    0.05       0  5016.1    0.05       0
  5020.1    0.05       0
Bank Sta=5016.1,5020.1
Exp/Cntr=0.3,0.1

Type RM Length L Ch R = 1,27790,498,498,498
BEGIN DESCRIPTION:
REED CREEK 57.0
END DESCRIPTION:
XS GIS Cut Line= 3
      2829305.65     10272203.11      2828996.00     10272161.00
      2828805.67     10272003.10
#Sta/Elev= 30
  4687.5 1287.55  4728.7 1281.59  4778.3 1272.14  4808.6 1265.11  4889.3 1255.10
  4939.8 1252.98  4970.6 1247.36  4990.2 1245.86  5011.4 1245.84  5011.7 1242.84
  5015.2 1242.84  5015.4 1245.84  5020.0 1246.83  5026.5 1246.35  5034.4 1248.46
  5040.9 1246.88  5055.2 1247.09  5083.9 1248.35  5104.7 1250.47  5112.5 1253.85
  5119.0 1252.73  5147.7 1257.93  5155.5 1260.65  5165.8 1261.47  5176.3 1263.04
  5182.8 1262.85  5197.1 1265.79  5240.1 1269.65  5244.0 1271.40  5247.3 1271.40
#Mann=5,-1,0
  4687.5    0.12       0  4970.6    0.05       0  5011.4    0.05       0
  5015.4    0.05       0  5165.8    0.12       0
Bank Sta=5011.4,5015.4
Exp/Cntr=0.3,0.1

Type RM Length L Ch R = 1,27292,369,369,369
BEGIN DESCRIPTION:
REED CREEK 56.0
END DESCRIPTION:
XS GIS Cut Line= 3
      2829355.69     10272003.13      2829188.00     10271730.00
      2828905.70     10271603.12
#Sta/Elev= 30
  4679.5 1277.28  4714.7 1271.93  4729.8 1267.99  4738.2 1267.27  4760.7 1261.65
  4766.5 1261.18  4781.9 1256.11  4803.2 1250.70  4809.1 1249.96  4876.7 1247.54
  4903.8 1245.17  4949.4 1243.32  4977.3 1241.54  4995.4 1239.00  4995.7 1236.00
  4999.2 1236.00  4999.4 1239.00  5024.0 1242.05  5035.4 1245.56  5052.6 1248.08
  5106.9 1252.72  5127.6 1254.30  5150.8 1258.28  5156.2 1257.75  5169.8 1259.11
  5248.9 1267.28  5265.7 1269.61  5272.0 1271.46  5287.6 1272.36  5309.5 1275.77
#Mann=5,-1,0
  4679.5    0.12       0  4995.4    0.07       0  4999.4    0.12       0
  5106.9    0.05       0  5169.8    0.12       0
Bank Sta=4995.4,4999.4
Exp/Cntr=0.3,0.1

Type RM Length L Ch R = 1,26923,480,480,480
BEGIN DESCRIPTION:
REED CREEK 55.0
END DESCRIPTION:
XS GIS Cut Line= 3
      2829505.64     10271453.12      2829445.50     10271466.00
      2829155.65     10271403.10
#Sta/Elev= 30
  4938.5 1251.25  4941.0 1251.25  4963.2 1246.23  4969.1 1239.24  4977.4 1233.39
  4977.6 1230.39  4981.1 1230.39  4981.4 1233.39  4997.3 1235.11  5002.5 1235.11
  5010.0 1237.61  5020.3 1238.05  5061.2 1238.39  5071.4 1237.38  5080.5 1238.50
  5091.9 1237.54  5102.1 1237.95  5112.4 1239.27  5122.6 1238.58  5129.6 1239.34
  5143.1 1239.44  5173.7 1241.19  5194.2 1241.15  5227.9 1243.10  5255.6 1245.65
  5265.9 1246.87  5272.0 1248.05  5277.1 1248.25  5294.0 1250.61  5296.6 1250.61
#Mann=3,-1,0
  4938.5    0.05       0  4977.4    0.05       0  4981.4    0.05       0
Bank Sta=4977.4,4981.4
Exp/Cntr=0.3,0.1

Type RM Length L Ch R = 1,26443,446,446,446
BEGIN DESCRIPTION:
REED CREEK 54.0
END DESCRIPTION:
XS GIS Cut Line= 3
      2829655.71     10271253.13      2829334.00     10271040.00
      2829205.67     10271053.11
#Sta/Elev= 30
  4614.1 1271.23  4617.1 1271.23  4621.7 1269.49  4636.7 1266.94  4663.8 1263.04
  4751.0 1252.40  4766.1 1249.87  4781.1 1248.51  4808.1 1243.66  4838.3 1242.00
  4844.2 1241.10  4853.3 1241.62  4874.4 1238.73  4880.3 1238.74  4910.5 1235.59
  4931.5 1234.58  4974.0 1230.76  5006.4 1226.89  5006.6 1223.89  5010.1 1223.89
  5010.4 1226.89  5038.5 1231.89  5048.6 1235.51  5058.6 1237.93  5076.7 1243.65
  5081.8 1242.35  5088.8 1244.76  5108.9 1248.97  5118.9 1252.50  5129.0 1254.10
#Mann=3,-1,0
  4614.1    0.05       0  5006.4    0.05       0  5010.4    0.05       0
Bank Sta=5006.4,5010.4
Exp/Cntr=0.3,0.1

Type RM Length L Ch R = 1,25997,397,397,397
BEGIN DESCRIPTION:
REED CREEK 53.0
END DESCRIPTION:
XS GIS Cut Line= 3
      2829405.69     10270553.11      2829331.50     10270601.00
      2829205.67     10270803.13
#Sta/Elev= 30
  4911.7 1240.82  4914.7 1240.82  4919.3 1238.32  4925.2 1236.46  4934.5 1232.63
  4940.4 1229.52  4955.6 1223.67  4981.1 1222.72  4981.4 1219.72  4984.9 1219.72
  4985.1 1222.72  4985.4 1222.74  4995.8 1223.65  5000.0 1223.83  5005.0 1225.30
  5035.7 1226.50  5041.6 1227.06  5056.9 1226.84  5062.8 1227.73  5072.3 1228.04
  5078.1 1228.84  5103.0 1230.66  5136.0 1233.25  5151.3 1235.02  5193.8 1238.57
  5209.2 1240.23  5215.0 1241.66  5224.5 1242.13  5235.1 1243.90  5238.1 1243.90
#Mann=6,-1,0
  4911.7    0.12       0  4981.1    0.07       0  4985.1    0.12       0
  4985.4    0.05       0  4995.8    0.12       0  5103.0    0.05       0
Bank Sta=4981.1,4985.1
Exp/Cntr=0.3,0.1

Type RM Length L Ch R = 1,25600,331,331,331
BEGIN DESCRIPTION:
Mapping XS 051ed89f
END DESCRIPTION:
XS GIS Cut Line= 3
      2829347.20     10270370.75      2829106.88     10270355.73
      2828716.33     10270641.12
#Sta/Elev= 30
  4609.6 1233.57  4654.0 1229.74  4731.4 1230.93  4885.6 1225.69  4906.4 1220.93
  4921.1 1221.18  4924.2 1218.58  4927.3 1215.97  4933.8 1214.94  4934.0 1211.94
  4937.5 1211.94  4937.8 1214.94  4942.0 1218.03  4950.4 1218.37  4956.6 1220.88
  4971.3 1218.33  5000.5 1217.13  5006.8 1215.12  5042.4 1217.60  5050.5 1216.46
  5071.7 1218.69  5092.5 1224.66  5107.2 1223.86  5142.7 1227.37  5222.3 1229.45
  5249.3 1233.65  5293.3 1231.41  5299.5 1232.83  5328.9 1228.31  5334.1 1229.29
#Mann=5,-1,0
  4609.6    0.05       0  4924.2    0.12       0  4933.8    0.07       0
  4937.8    0.12       0  5050.5    0.05       0
Bank Sta=4933.8,4937.8
Exp/Cntr=0.3,0.1

Type RM Length L Ch R = 1,25269,678,678,678
BEGIN DESCRIPTION:
Mapping XS c379caa9
END DESCRIPTION:
XS GIS Cut Line= 3
      2829197.01     10270265.60      2828506.02     10270235.55
      2828205.61     10270070.33
#Sta/Elev= 30
  4555.0 1220.33  4616.4 1219.53  4656.4 1220.53  4696.5 1219.33  4716.5 1220.62
  4729.4 1218.98  4736.5 1219.98  4796.6 1217.64  4889.1 1217.33  4926.7 1217.17
  5001.5 1210.81  5014.8 1209.68  5015.0 1206.68  5018.5 1206.68  5018.8 1209.68
  5036.8 1213.23  5066.8 1215.18  5116.9 1212.91  5166.9 1215.74  5176.9 1215.08
  5217.0 1219.57  5366.4 1230.43  5372.6 1232.08  5388.1 1231.70  5406.1 1233.47
  5516.2 1245.19  5543.8 1249.21  5551.0 1251.32  5566.6 1251.26  5589.5 1253.27
#Mann=7,-1,0
  4555.0    0.05       0  4889.1    0.12       0  5001.5    0.05       0
  5014.8    0.07       0  5018.8    0.05       0  5406.1    0.12       0
  5516.2    0.05       0
Bank Sta=5014.8,5018.8
Exp/Cntr=0.3,0.1

Type RM Length L Ch R = 1,24591,463,463,463
BEGIN DESCRIPTION:
REED CREEK 50.0
END DESCRIPTION:
XS GIS Cut Line= 3
      2829405.67     10270253.09      2829317.50     10270090.00
      2829255.68     10269953.11
#Sta/Elev= 30
  4814.6 1230.56  4817.4 1230.56  4822.7 1227.79  4828.4 1227.77  4844.6 1221.69
  4850.2 1221.79  4866.4 1217.22  4872.1 1216.93  4882.6 1213.78  4888.3 1214.04
  4916.9 1208.71  4926.4 1207.82  4931.2 1208.57  4954.0 1205.91  4962.4 1204.36
  4970.2 1201.16  4990.0 1198.57  4990.3 1195.57  4993.8 1195.57  4994.0 1198.57
  4996.7 1199.93  5014.8 1201.64  5043.4 1203.12  5061.0 1205.89  5066.5 1206.05
  5084.2 1209.63  5089.7 1209.72  5095.3 1211.16  5117.3 1213.33  5150.2 1217.83
#Mann=5,-1,0
  4814.6    0.05       0  4931.2    0.12       0  4990.0    0.07       0
  4994.0    0.12       0  5117.3    0.05       0
Bank Sta=4990,4994
Exp/Cntr=0.3,0.1

Type RM Length L Ch R = 1,24128,457,457,457
BEGIN DESCRIPTION:
REED CREEK 49.0
END DESCRIPTION:
XS GIS Cut Line= 3
      2829655.68     10270053.10      2829592.00     10269754.00
      2829355.64     10269653.09
#Sta/Elev= 30
  4694.2 1227.11  4724.9 1221.14  4786.2 1213.73  4806.6 1210.54  4818.1 1207.43
  4857.5 1202.35  4862.6 1199.84  4868.0 1198.53  4907.0 1196.64  4919.1 1195.22
  4956.6 1194.66  4961.7 1193.15  4990.7 1191.12  4995.9 1189.64  4996.1 1186.64
  4999.6 1186.64  4999.9 1189.64  5013.7 1191.30  5019.1 1190.71  5029.7 1191.51
  5072.1 1196.76  5083.0 1196.53  5095.3 1198.07  5119.0 1198.41  5137.1 1200.51
  5166.2 1201.03  5202.6 1206.50  5247.9 1210.92  5254.2 1213.19  5257.0 1213.19
#Mann=4,-1,0
  4694.2    0.12       0  4995.9    0.07       0  4999.9    0.12       0
  5029.7    0.05       0
Bank Sta=4995.9,4999.9
Exp/Cntr=0.3,0.1

Type RM Length L Ch R = 1,23671,498,498,498
BEGIN DESCRIPTION:
REED CREEK 48.0
END DESCRIPTION:
XS GIS Cut Line= 3
      2829905.68     10269953.11      2829920.50     10269904.00
      2829955.68     10269753.15
#Sta/Elev= 28
  4948.7 1200.43  4951.3 1200.43  4965.2 1191.85  4970.4 1188.90  4980.0 1183.14
  4990.5 1180.59  4995.9 1177.46  4996.1 1174.46  4999.6 1174.46  4999.9 1177.46
  5003.4 1177.48  5011.2 1178.61  5021.4 1178.42  5031.7 1180.43  5040.8 1181.87
  5046.0 1183.15  5052.3 1184.91  5083.1 1190.63  5088.5 1192.99  5093.7 1193.65
  5103.6 1195.09  5113.9 1197.39  5124.1 1198.26  5131.1 1199.55  5136.2 1199.69
  5144.7 1201.99  5152.4 1203.67  5154.9 1203.67
#Mann=3,-1,0
  4948.7    0.12       0  4995.9    0.07       0  4999.9    0.12       0
Bank Sta=4995.9,4999.9
Exp/Cntr=0.3,0.1

Type RM Length L Ch R = 1,23173,476,476,476
BEGIN DESCRIPTION:
REED CREEK 47.0
END DESCRIPTION:
XS GIS Cut Line= 3
      2830405.68     10270253.10      2830407.25     10269993.00
      2830305.68     10269603.11
#Sta/Elev= 30
  4739.9 1222.18  4742.4 1222.18  4749.9 1219.73  4759.9 1218.21  4769.9 1215.11
  4789.9 1210.95  4819.9 1206.96  4845.5 1201.97  4889.9 1193.86  4919.9 1189.99
  4929.9 1186.29  4949.9 1181.00  4989.9 1173.82  5028.1 1172.78  5039.2 1172.28
  5039.5 1169.28  5043.0 1169.28  5043.2 1172.28  5100.4 1178.04  5175.6 1183.31
  5216.9 1187.32  5258.2 1192.68  5304.2 1198.81  5309.9 1200.84  5344.7 1205.56
  5361.6 1210.26  5380.1 1212.60  5392.6 1215.30  5400.3 1217.88  5402.9 1217.88
#Mann=6,-1,0
  4739.9    0.12       0  4845.5    0.05       0  5028.1    0.12       0
  5039.2    0.05       0  5043.2    0.12       0  5100.4    0.05       0
Bank Sta=5039.2,5043.2
Exp/Cntr=0.3,0.1

Type RM Length L Ch R = 1,22697,466,466,466
BEGIN DESCRIPTION:
REED CREEK 46.0
END DESCRIPTION:
XS GIS Cut Line= 3
      2830905.67     10269853.10      2830820.25     10269766.00
      2830505.65     10269503.08
#Sta/Elev= 30
  4878.0 1176.52  4881.5 1176.52  4885.1 1175.72  4899.2 1174.30  4920.3 1173.04
  4948.6 1170.33  4969.9 1167.47  4984.1 1164.19  4991.1 1163.27  4996.2 1163.25
  4996.4 1160.25  5000.0 1160.25  5000.3 1163.25  5012.4 1163.71  5026.7 1164.83
  5033.2 1165.78  5076.2 1168.06  5104.8 1170.98  5136.8 1173.11  5168.5 1176.42
  5175.4 1177.60  5189.4 1178.51  5232.3 1184.56  5296.1 1191.89  5310.4 1194.51
  5331.8 1197.19  5353.3 1198.94  5382.0 1203.85  5406.7 1209.08  5410.0 1209.08
#Mann=5,-1,0
  4878.0    0.05       0  4899.2    0.12       0  4996.2    0.07       0
  5000.3    0.12       0  5136.8    0.05       0
Bank Sta=4996.2,5000.3
Exp/Cntr=0.3,0.1

Type RM Length L Ch R = 1,22231,463,463,463
BEGIN DESCRIPTION:
REED CREEK 45.0
END DESCRIPTION:
XS GIS Cut Line= 3
      2831155.68     10269953.12      2831234.75     10269555.00
      2831205.67     10269453.07
#Sta/Elev= 30
  4594.1 1181.19  4619.7 1178.57  4670.8 1175.06  4722.0 1171.71  4736.8 1171.60
  4778.3 1168.26  4849.0 1164.94  4880.6 1161.99  4900.0 1161.34  4920.4 1161.81
  4940.8 1160.38  4961.1 1160.21  4971.3 1159.91  4977.8 1159.06  4982.9 1159.24
  4991.7 1157.43  4996.4 1155.05  4996.6 1152.05  5000.2 1152.05  5000.5 1155.05
  5022.8 1155.36  5033.2 1159.78  5046.9 1167.90  5050.0 1169.76  5055.2 1169.00
  5064.4 1171.24  5083.8 1174.21  5089.0 1174.36  5095.6 1175.71  5106.0 1175.95
#Mann=4,-1,0
  4594.1    0.05       0  4996.4    0.05       0  5000.5    0.05       0
  5046.9    0.12       0
Bank Sta=4996.4,5000.5
Exp/Cntr=0.3,0.1

Type RM Length L Ch R = 1,21768,400,400,400
BEGIN DESCRIPTION:
REED CREEK 44.0
END DESCRIPTION:
XS GIS Cut Line= 3
      2831755.70     10269703.15      2831668.25     10269494.00
      2831555.71     10269353.14
#Sta/Elev= 30
  4773.3 1167.91  4788.0 1166.95  4805.9 1164.89  4817.2 1162.79  4827.5 1162.13
  4841.0 1159.82  4864.8 1154.64  4870.9 1152.41  4881.7 1149.63  4894.0 1147.15
  4912.4 1147.82  4917.8 1148.83  4925.1 1149.14  4941.6 1147.87  4965.4 1147.94
  4995.6 1144.53  4995.9 1141.53  4999.7 1141.53  5000.0 1144.53  5003.8 1144.53
  5024.2 1150.22  5045.0 1154.23  5070.4 1155.78  5109.1 1160.66  5123.5 1161.61
  5144.3 1164.63  5152.3 1166.42  5158.7 1166.65  5166.7 1168.87  5180.3 1170.33
#Mann=4,-1,0
  4773.3    0.12       0  4995.6    0.07       0  5000.0    0.12       0
  5070.4    0.05       0
Bank Sta=4995.6,5000
Exp/Cntr=0.3,0.1

Type RM Length L Ch R = 1,21368,439,439,439
BEGIN DESCRIPTION:
REED CREEK 43.0
END DESCRIPTION:
XS GIS Cut Line= 3
      2832205.67     10269753.08      2832025.25     10269338.00
      2831955.65     10269253.07
#Sta/Elev= 30
  4547.4 1178.41  4561.8 1177.50  4579.8 1174.72  4585.3 1175.29  4608.7 1170.96
  4637.6 1168.60  4645.9 1166.91  4684.5 1160.87  4736.8 1156.63  4760.3 1152.53
  4765.7 1153.53  4778.3 1152.18  4783.7 1150.63  4789.2 1152.60  4820.0 1148.08
  4911.9 1142.99  4970.4 1137.37  4970.7 1134.37  4974.5 1134.37  4974.9 1137.37
  5010.0 1139.07  5017.9 1144.56  5024.3 1144.25  5038.7 1151.37  5073.9 1155.26
  5081.8 1157.60  5088.2 1156.79  5102.6 1158.85  5106.5 1160.99  5109.8 1160.99
#Mann=6,-1,0
  4547.4    0.05       0  4645.9    0.12       0  4778.3    0.05       0
  4970.4    0.05       0  4974.9    0.05       0  5102.6    0.12       0
Bank Sta=4970.4,4974.9
Exp/Cntr=0.3,0.1

Type RM Length L Ch R = 1,20929,457,457,457
BEGIN DESCRIPTION:
REED CREEK 42.0
END DESCRIPTION:
XS GIS Cut Line= 3
      2832455.69     10269403.14      2832428.75     10269219.00
      2832205.66     10269103.10
#Sta/Elev= 30
  4813.9 1154.61  4824.0 1154.60  4834.1 1151.65  4843.8 1150.14  4848.9 1150.48
  4854.4 1148.91  4884.7 1144.98  4913.7 1143.13  4918.8 1141.54  4935.2 1139.53
  4945.3 1137.12  4965.5 1130.53  4981.4 1128.51  4981.7 1125.51  4985.6 1125.51
  4985.9 1128.51  4995.0 1129.04  5014.7 1130.16  5027.6 1132.97  5078.2 1136.20
  5116.1 1143.97  5119.9 1144.09  5126.9 1144.31  5138.7 1146.80  5154.7 1147.06
  5176.8 1148.49  5193.3 1150.76  5198.9 1150.34  5215.4 1152.15  5251.4 1154.04
#Mann=6,-1,0
  4813.9    0.05       0  4981.4    0.07       0  4985.9    0.05       0
  4995.0    0.12       0  5078.2    0.05       0  5119.9    0.12       0
Bank Sta=4981.4,4985.9
Exp/Cntr=0.3,0.1

Type RM Length L Ch R = 1,20472,475,475,475
BEGIN DESCRIPTION:
REED CREEK 41.0
END DESCRIPTION:
XS GIS Cut Line= 3
      2832805.69     10269303.11      2832849.25     10269048.00
      2832805.69     10268953.12
#Sta/Elev= 30
  4741.2 1147.54  4751.3 1145.71  4773.8 1143.84  4791.9 1141.32  4812.2 1140.03
  4828.9 1137.63  4833.9 1138.14  4846.1 1136.08  4889.0 1130.70  4894.1 1131.01
  4913.7 1129.03  4944.1 1123.89  4949.1 1124.24  4954.2 1122.39  4963.8 1122.89
  4984.7 1121.30  4992.4 1119.01  4992.8 1116.01  4996.9 1116.01  4997.2 1119.01
  4999.9 1122.34  5005.4 1122.34  5015.7 1125.34  5021.2 1124.38  5027.4 1128.32
  5038.4 1130.47  5049.7 1130.49  5067.2 1133.01  5072.7 1133.06  5104.4 1136.78
#Mann=5,-1,0
  4741.2    0.12       0  4846.1    0.05       0  4963.8    0.12       0
  4992.4    0.07       0  4997.2    0.12       0
Bank Sta=4992.4,4997.2
Exp/Cntr=0.3,0.1

Type RM Length L Ch R = 1,19997,391,391,391
BEGIN DESCRIPTION:
REED CREEK 40.0
END DESCRIPTION:
XS GIS Cut Line= 3
      2833305.68     10269103.15      2833309.50     10268947.00
      2833155.69     10268853.11
#Sta/Elev= 30
  4843.8 1132.17  4846.3 1132.17  4854.0 1130.75  4863.8 1129.39  4893.9 1122.88
  4923.9 1118.34  4933.9 1116.99  4952.2 1117.11  4973.9 1117.63  4983.9 1116.68
  4991.4 1115.38  4991.8 1112.38  4995.9 1112.38  4996.3 1115.38  4999.4 1115.99
  5013.7 1116.11  5019.6 1117.53  5035.0 1119.09  5040.9 1120.49  5058.2 1121.92
  5086.5 1124.62  5108.5 1125.41  5121.6 1127.44  5135.7 1128.13  5145.1 1129.08
  5150.0 1129.02  5157.0 1130.33  5166.6 1130.38  5172.5 1131.13  5180.2 1131.01
#Mann=7,-1,0
  4843.8    0.12       0  4854.0    0.05       0  4952.2    0.12       0
  4991.4    0.07       0  4996.3    0.12       0  5058.2    0.05       0
  5150.0    0.12       0
Bank Sta=4991.4,4996.3
Exp/Cntr=0.3,0.1

Type RM Length L Ch R = 1,19606,490,490,490
BEGIN DESCRIPTION:
REED CREEK 39.0
END DESCRIPTION:
XS GIS Cut Line= 3
      2833555.67     10269053.14      2833673.75     10268808.00
      2833805.68     10268503.12
#Sta/Elev= 30
  4727.9 1127.93  4804.6 1121.23  4877.7 1116.66  4938.8 1115.30  4945.6 1113.83
  4961.0 1113.13  4968.2 1111.52  4973.8 1111.83  4997.4 1109.94  4997.8 1106.94
  5002.0 1106.94  5002.4 1109.94  5014.1 1111.18  5019.6 1110.39  5037.6 1112.05
  5048.9 1111.45  5098.1 1113.56  5113.5 1115.10  5119.0 1114.47  5136.1 1118.05
  5142.4 1121.98  5147.9 1121.56  5157.9 1125.71  5194.9 1127.24  5218.4 1131.10
  5247.3 1133.49  5265.3 1136.45  5270.8 1136.06  5299.7 1140.80  5332.2 1144.24
#Mann=5,-1,0
  4727.9    0.12       0  4804.6    0.05       0  4997.4    0.05       0
  5002.4    0.05       0  5098.1    0.12       0
Bank Sta=4997.4,5002.4
Exp/Cntr=0.3,0.1

Type RM Length L Ch R = 1,19116,443,443,443
BEGIN DESCRIPTION:
REED CREEK 38.0
END DESCRIPTION:
XS GIS Cut Line= 3
      2834055.68     10269303.14      2834081.00     10269028.00
      2834005.69     10268703.12
#Sta/Elev= 30
  4723.7 1124.06  4844.2 1112.64  4883.4 1109.35  4888.4 1109.37  4904.5 1107.63
  4924.8 1106.60  4974.8 1103.54  4984.8 1103.55  4993.2 1102.12  4995.7 1100.69
  4996.1 1097.69  5000.4 1097.69  5000.7 1100.69  5015.3 1100.83  5043.3 1106.43
  5048.4 1105.61  5086.0 1109.49  5091.1 1108.50  5094.1 1108.88  5117.9 1112.30
  5133.8 1113.99  5138.9 1113.75  5159.0 1115.84  5219.7 1119.51  5261.6 1123.27
  5266.9 1124.54  5282.2 1125.54  5288.7 1126.86  5314.7 1130.61  5333.5 1131.68
#Mann=7,-1,0
  4723.7    0.05       0  4924.8    0.12       0  4995.7    0.07       0
  5000.7    0.12       0  5094.1    0.05       0  5219.7    0.12       0
  5288.7    0.05       0
Bank Sta=4995.7,5000.7
Exp/Cntr=0.3,0.1

Type RM Length L Ch R = 1,18673,463,463,463
BEGIN DESCRIPTION:
REED CREEK 37.0
END DESCRIPTION:
XS GIS Cut Line= 3
      2834505.69     10269103.14      2834472.25     10268877.00
      2834355.71     10268703.15
#Sta/Elev= 30
  4771.4 1111.11  4822.0 1107.30  4929.4 1101.23  4953.4 1100.76  4963.5 1099.16
  4983.7 1098.00  4993.8 1096.72  4999.4 1097.40  5015.7 1096.73  5019.3 1096.13
  5019.6 1093.13  5023.9 1093.13  5024.3 1096.13  5028.8 1096.78  5042.8 1097.29
  5057.8 1096.98  5064.9 1097.50  5074.3 1099.78  5087.8 1103.17  5093.8 1103.64
  5114.8 1109.60  5129.8 1111.51  5136.7 1111.89  5144.8 1112.57  5150.8 1114.10
  5159.8 1114.63  5165.8 1115.81  5180.8 1116.37  5206.3 1119.60  5209.3 1119.60
#Mann=6,-1,0
  4771.4    0.05       0  4929.4    0.12       0  5019.3    0.07       0
  5024.3    0.12       0  5074.3    0.05       0  5136.7    0.12       0
Bank Sta=5019.3,5024.3
Exp/Cntr=0.3,0.1

Type RM Length L Ch R = 1,18210,489,489,489
BEGIN DESCRIPTION:
REED CREEK 36.0
END DESCRIPTION:
XS GIS Cut Line= 3
      2834805.67     10269003.13      2834927.50     10268796.00
      2834905.69     10268603.13
#Sta/Elev= 30
  4759.7 1104.64  4840.9 1100.93  4927.7 1097.58  4943.3 1095.92  4949.1 1095.80
  4964.8 1093.26  4970.6 1093.61  4980.1 1091.24  4986.3 1089.15  4989.5 1089.09
  4989.9 1086.09  4994.2 1086.09  4994.6 1089.09  4998.8 1089.69  5004.0 1089.69
  5013.0 1091.70  5023.0 1091.52  5031.6 1090.81  5043.2 1090.36  5053.2 1090.66
  5059.5 1093.83  5064.5 1093.69  5073.4 1094.32  5143.8 1100.12  5149.2 1101.50
  5154.3 1100.95  5163.9 1102.50  5174.0 1104.93  5185.4 1106.98  5194.1 1106.77
#Mann=5,-1,0
  4759.7    0.05       0  4989.5    0.05       0  4994.6    0.05       0
  5031.6    0.12       0  5185.4    0.05       0
Bank Sta=4989.5,4994.6
Exp/Cntr=0.3,0.1

Type RM Length L Ch R = 1,17721,478,478,478
BEGIN DESCRIPTION:
REED CREEK 35.0
END DESCRIPTION:
XS GIS Cut Line= 3
      2835155.66     10269053.13      2835390.50     10268899.00
      2835455.69     10268753.10
#Sta/Elev= 30
  4719.1 1099.58  4726.7 1099.18  4732.7 1100.07  4777.9 1099.09  4790.9 1098.25
  4814.1 1095.72  4820.1 1094.43  4835.2 1093.75  4841.2 1094.07  4922.5 1090.61
  4934.6 1089.17  4943.7 1088.68  4958.4 1086.24  4979.8 1084.73  4991.5 1082.85
  4991.9 1079.85  4996.3 1079.85  4996.7 1082.85  5029.4 1086.75  5047.1 1090.30
  5052.6 1092.30  5061.2 1093.75  5070.3 1093.23  5075.8 1094.52  5083.1 1093.99
  5099.0 1094.71  5105.0 1095.89  5122.2 1098.00  5137.9 1098.76  5159.8 1100.63
#Mann=3,-1,0
  4719.1    0.12       0  4991.5    0.07       0  4996.7    0.12       0
Bank Sta=4991.5,4996.7
Exp/Cntr=0.3,0.1

Type RM Length L Ch R = 1,17243,471,471,471
BEGIN DESCRIPTION:
REED CREEK 34.0
END DESCRIPTION:
XS GIS Cut Line= 3
      2835855.67     10269403.07      2835776.00     10269177.00
      2835655.68     10268803.08
#Sta/Elev= 30
  4760.3 1105.08  4765.1 1104.86  4806.7 1098.73  4823.9 1095.15  4832.3 1092.52
  4837.6 1092.71  4845.1 1090.96  4883.7 1087.79  4894.2 1086.46  4899.5 1086.92
  4919.3 1085.21  4925.2 1083.41  4930.5 1083.33  4950.8 1079.14  4969.1 1077.85
  4969.6 1074.85  4975.1 1074.85  4975.6 1077.85  4987.1 1079.27  5025.1 1080.78
  5045.4 1082.53  5050.7 1081.68  5077.5 1084.22  5082.8 1083.41  5088.1 1084.89
  5114.8 1087.31  5120.1 1086.73  5211.1 1091.48  5290.8 1093.67  5392.8 1096.35
#Mann=6,-1,0
  4760.3    0.12       0  4765.1    0.05       0  4883.7    0.12       0
  4969.1    0.07       0  4975.6    0.12       0  5290.8    0.05       0
Bank Sta=4969.1,4975.6
Exp/Cntr=0.3,0.1

Type RM Length L Ch R = 1,16772,486,486,486
BEGIN DESCRIPTION:
REED CREEK 33.0
END DESCRIPTION:
XS GIS Cut Line= 3
      2836255.67     10269153.09      2836185.75     10269031.00
      2835955.68     10268953.11
#Sta/Elev= 30
  4859.3 1091.01  4867.2 1090.99  4882.3 1089.43  4888.8 1086.31  4897.1 1084.62
  4904.6 1083.16  4916.9 1081.40  4931.9 1079.68  4939.5 1079.49  4963.0 1076.93
  4969.4 1075.99  4975.1 1075.54  4985.2 1075.42  4987.7 1074.65  4988.2 1071.65
  4993.7 1071.65  4994.2 1074.65  4995.9 1076.27  5002.7 1076.27  5007.2 1076.99
  5021.2 1075.91  5031.7 1075.88  5039.9 1076.47  5052.9 1078.64  5070.0 1080.80
  5101.5 1082.40  5195.8 1084.83  5211.2 1085.01  5227.2 1085.91  5242.9 1086.01
#Mann=6,-1,0
  4859.3    0.12       0  4897.1    0.05       0  4939.5    0.12       0
  4987.7    0.07       0  4994.2    0.12       0  5039.9    0.05       0
Bank Sta=4987.7,4994.2
Exp/Cntr=0.3,0.1

Type RM Length L Ch R = 1,16286,398,398,398
BEGIN DESCRIPTION:
REED CREEK 32.0
END DESCRIPTION:
XS GIS Cut Line= 3
      2836405.67     10268703.08      2836324.75     10268575.00
      2836055.71     10268603.11
#Sta/Elev= 30
  4848.5 1079.80  4877.3 1078.50  4892.6 1077.23  4907.6 1077.19  4913.8 1075.96
  4919.7 1076.19  4943.1 1072.55  4956.1 1071.30  4965.5 1071.20  4983.4 1069.37
  4983.9 1066.37  4989.4 1066.37  4989.9 1069.37  5020.3 1069.98  5027.1 1069.57
  5032.1 1070.91  5039.3 1070.77  5059.4 1071.78  5069.4 1071.49  5079.5 1070.39
  5099.6 1069.81  5109.7 1070.28  5125.5 1071.96  5130.5 1072.10  5149.9 1074.26
  5210.2 1077.69  5218.8 1078.73  5223.8 1078.85  5230.3 1080.08  5270.5 1080.92
#Mann=4,-1,0
  4848.5    0.12       0  4983.4    0.07       0  4989.9    0.12       0
  5020.3    0.05       0
Bank Sta=4983.4,4989.9
Exp/Cntr=0.3,0.1

Type RM Length L Ch R = 1,15888,423,423,423
BEGIN DESCRIPTION:
REED CREEK 31.0
END DESCRIPTION:
XS GIS Cut Line= 3
      2836705.71     10268453.15      2836598.75     10268287.00
      2836505.66     10268153.08
#Sta/Elev= 30
  4802.4 1078.84  4805.4 1078.84  4810.0 1077.94  4831.2 1077.02  4861.5 1074.71
  4882.7 1073.79  4897.6 1072.41  4903.8 1071.37  4909.7 1071.39  4919.4 1070.65
  4940.1 1069.17  4955.3 1067.07  4961.2 1065.74  4968.9 1063.42  4973.1 1062.85
  4973.6 1059.85  4979.3 1059.85  4979.8 1062.85  5041.3 1064.26  5048.3 1065.68
  5054.4 1065.68  5069.2 1067.19  5077.8 1068.65  5119.8 1072.17  5134.7 1076.09
  5140.8 1076.41  5149.5 1078.23  5155.6 1078.07  5160.0 1079.57  5163.1 1079.57
#Mann=4,-1,0
  4802.4    0.05       0  4919.4    0.12       0  4973.1    0.07       0
  4979.8    0.12       0
Bank Sta=4973.1,4979.8
Exp/Cntr=0.3,0.1

Type RM Length L Ch R = 1,15465,497,497,497
BEGIN DESCRIPTION:
REED CREEK 30.0
END DESCRIPTION:
XS GIS Cut Line= 3
      2836955.68     10268303.10      2836970.25     10268090.00
      2836755.68     10268003.11
#Sta/Elev= 30
  4786.4 1073.56  4846.5 1070.18  4855.6 1069.30  4860.6 1069.55  4876.6 1068.95
  4926.7 1064.24  4956.8 1062.19  4966.8 1060.74  4986.9 1058.73  5002.5 1059.39
  5004.3 1057.98  5004.8 1054.98  5010.6 1054.98  5011.1 1057.98  5026.4 1058.55
  5031.8 1059.35  5037.3 1061.27  5055.9 1064.08  5073.2 1065.00  5080.0 1065.27
  5085.4 1066.20  5102.0 1066.71  5114.9 1067.90  5139.0 1068.79  5145.2 1069.69
  5163.1 1070.79  5199.1 1072.65  5209.9 1072.73  5216.7 1073.39  5231.5 1073.75
#Mann=4,-1,0
  4786.4    0.05       0  5004.3    0.05       0  5011.1    0.05       0
  5073.2    0.12       0
Bank Sta=5004.3,5011.1
Exp/Cntr=0.3,0.1

Type RM Length L Ch R = 1,14968,489,489,489
BEGIN DESCRIPTION:
REED CREEK 29.0
END DESCRIPTION:
XS GIS Cut Line= 3
      2837355.69     10268253.10      2837421.50     10267993.00
      2837405.68     10267853.09
#Sta/Elev= 30
  4731.7 1071.00  4754.8 1070.28  4790.6 1067.64  4836.8 1066.17  4845.2 1065.30
  4877.8 1064.47  4907.0 1062.87  4913.7 1061.96  4918.8 1062.11  4954.7 1056.85
  4968.9 1055.85  4979.3 1056.30  4989.6 1055.13  4992.1 1054.28  4992.6 1051.28
  4998.9 1051.28  4999.4 1054.28  5000.8 1054.32  5002.5 1054.36  5006.1 1055.99
  5011.1 1055.49  5020.0 1057.39  5040.1 1059.35  5050.2 1061.23  5080.4 1064.93
  5095.9 1067.99  5110.6 1069.33  5120.7 1071.39  5130.7 1072.80  5140.8 1073.51
#Mann=4,-1,0
  4731.7    0.05       0  4992.1    0.05       0  4999.4    0.05       0
  5000.8    0.12       0
Bank Sta=4992.1,4999.4
Exp/Cntr=0.3,0.1

Type RM Length L Ch R = 1,14479,961,961,961
BEGIN DESCRIPTION:
REED CREEK 28.0
END DESCRIPTION:
XS GIS Cut Line= 3
      2837455.69     10268553.10      2837876.50     10268136.00
      2837905.68     10267353.14
#Sta/Elev= 30
  4407.5 1083.08  4435.7 1080.52  4464.0 1079.37  4500.5 1075.32  4598.4 1069.05
  4640.8 1068.08  4669.1 1065.87  4782.3 1061.32  4874.2 1059.61  4901.8 1058.21
  4959.0 1056.66  4987.3 1053.40  4998.5 1050.78  5019.3 1048.94  5019.8 1045.94
  5026.1 1045.94  5026.6 1048.94  5032.9 1049.10  5042.9 1051.31  5052.9 1055.43
  5072.9 1059.52  5082.9 1063.02  5110.1 1065.01  5223.0 1065.77  5283.1 1064.59
  5343.1 1061.68  5384.5 1060.69  5413.2 1063.58  5533.3 1068.28  5783.4 1082.52
#Mann=5,-1,0
  4407.5    0.05       0  4500.5    0.12       0  4901.8    0.05       0
  5019.3    0.05       0  5026.6    0.05       0
Bank Sta=5019.3,5026.6
Exp/Cntr=0.3,0.1

Type RM Length L Ch R = 1,13518,264,264,264
BEGIN DESCRIPTION:
REED CREEK 27.0
END DESCRIPTION:
XS GIS Cut Line= 3
      2838555.65     10268503.08      2838462.25     10268407.00
      2838055.71     10268203.12
#Sta/Elev= 30
  4866.0 1061.40  4869.4 1061.40  4880.0 1060.49  4887.2 1061.67  4901.3 1058.33
  4925.1 1054.23  4936.6 1052.35  4943.8 1052.11  4950.7 1049.52  4964.9 1046.67
  4979.0 1045.37  4982.5 1044.26  4983.0 1041.26  4989.4 1041.26  4989.9 1044.26
  5016.4 1045.78  5029.7 1045.54  5044.3 1046.99  5061.1 1050.13  5074.5 1051.51
  5083.4 1050.23  5096.8 1050.82  5105.7 1050.14  5128.1 1053.40  5245.4 1055.35
  5262.1 1056.48  5275.8 1056.52  5329.2 1058.96  5396.2 1060.30  5454.8 1060.73
#Mann=5,-1,0
  4866.0    0.05       0  4869.4    0.12       0  4925.1    0.05       0
  4982.5    0.05       0  4989.9    0.05       0
Bank Sta=4982.5,4989.9
Exp/Cntr=0.3,0.1

Type RM Length L Ch R = 1,13254,1162,1162,1162
BEGIN DESCRIPTION:
Mapping XS 5968f8f4
END DESCRIPTION:
XS GIS Cut Line= 4
      2838810.75     10268478.06      2838630.48     10268207.66
      2838390.14     10268057.44      2838194.85     10267802.06
#Sta/Elev= 30
  4615.5 1055.79  4780.8 1057.26  4868.6 1056.50  4904.0 1056.55  4933.9 1054.60
  4940.0 1051.18  4946.3 1050.36  4955.3 1047.33  4976.5 1043.34  4997.7 1043.41
  5005.1 1044.90  5024.7 1042.97  5025.2 1039.97  5031.6 1039.97  5032.1 1042.97
  5049.6 1043.77  5061.2 1045.30  5099.4 1048.96  5149.8 1048.82  5165.2 1049.90
  5171.1 1049.13  5293.7 1052.13  5316.5 1051.55  5322.8 1053.41  5351.8 1053.17
  5366.4 1051.94  5451.6 1053.92  5466.1 1051.91  5480.6 1051.81  5545.4 1055.21
#Mann=5,-1,0
  4615.5    0.05       0  4868.6    0.12       0  5024.7    0.07       0
  5032.1    0.12       0  5061.2    0.05       0
Bank Sta=5024.7,5032.1
Exp/Cntr=0.3,0.1

Type RM Length L Ch R = 1,12092,499,499,499
BEGIN DESCRIPTION:
REED CREEK 25.0
END DESCRIPTION:
XS GIS Cut Line= 3
      2838755.70     10268103.09      2839178.75     10267451.00
      2839305.69     10267203.11
#Sta/Elev= 30
  4222.7 1053.93  4317.9 1048.66  4402.3 1046.74  4692.4 1044.33  4894.7 1043.79
  4915.8 1042.52  4925.0 1039.60  4931.0 1039.58  4946.1 1033.87  4952.1 1035.05
  4961.3 1033.40  4969.8 1033.30  4970.3 1030.30  4976.9 1030.30  4977.4 1033.30
  5020.1 1035.88  5025.9 1037.22  5048.2 1037.12  5053.8 1038.03  5070.4 1038.28
  5114.8 1036.44  5131.4 1039.56  5137.0 1038.90  5153.6 1043.23  5159.2 1041.83
  5175.8 1045.12  5181.4 1044.39  5198.0 1047.31  5203.6 1046.98  5278.5 1051.70
#Mann=3,-1,0
  4222.7    0.05       0  4969.8    0.03       0  4977.4    0.05       0
Bank Sta=4969.8,4977.4
Exp/Cntr=0.3,0.1

Type RM Length L Ch R = 1,11593,495,495,495
BEGIN DESCRIPTION:
REED CREEK 24.0
END DESCRIPTION:
XS GIS Cut Line= 3
      2839455.67     10267703.13      2839640.50     10267507.00
      2839705.66     10267403.15
#Sta/Elev= 30
  4730.5 1041.54  4808.4 1040.45  4850.9 1041.11  4857.8 1040.38  4865.1 1040.45
  4871.9 1039.85  4886.1 1039.77  4900.2 1039.98  4914.4 1040.65  4928.6 1040.46
  4950.0 1035.69  4964.1 1033.95  4977.9 1031.01  4985.2 1030.69  4988.2 1029.94
  4988.7 1026.94  4995.4 1026.94  4995.9 1029.94  4999.2 1030.46  5005.4 1030.30
  5014.8 1031.99  5020.7 1032.26  5028.2 1033.13  5036.0 1032.85  5041.9 1033.52
  5057.3 1033.54  5063.6 1034.41  5078.5 1037.80  5093.8 1043.16  5122.6 1045.25
#Mann=3,-1,0
  4730.5    0.05       0  4988.2    0.03       0  4995.9    0.05       0
Bank Sta=4988.2,4995.9
Exp/Cntr=0.3,0.1

Type RM Length L Ch R = 1,11098,474,474,474
BEGIN DESCRIPTION:
REED CREEK 23.0
END DESCRIPTION:
XS GIS Cut Line= 3
      2840155.67     10267953.08      2840049.50     10267663.00
      2840005.68     10267553.11
#Sta/Elev= 30
  4691.1 1048.60  4714.0 1047.20  4736.8 1046.29  4762.0 1043.48  4767.4 1043.68
  4776.3 1042.47  4786.9 1041.97  4792.6 1040.78  4817.4 1039.62  4840.1 1038.39
  4848.3 1036.78  4853.6 1037.25  4861.4 1035.43  4904.0 1031.54  4909.3 1031.79
  4914.7 1030.46  4947.2 1028.87  4965.0 1027.70  4995.6 1027.75  5010.6 1026.56
  5025.3 1026.74  5026.0 1026.25  5026.5 1023.25  5037.9 1023.25  5038.4 1026.25
  5042.9 1027.05  5049.6 1027.14  5054.2 1029.34  5086.0 1036.99  5118.3 1038.64
#Mann=7,-1,0
  4691.1    0.05       0  4714.0    0.12       0  4817.4    0.05       0
  4947.2    0.12       0  5026.0    0.07       0  5038.4    0.12       0
  5054.2    0.05       0
Bank Sta=5026,5038.4
Exp/Cntr=0.3,0.1

Type RM Length L Ch R = 1,10624,448,448,448
BEGIN DESCRIPTION:
REED CREEK 22.0
END DESCRIPTION:
XS GIS Cut Line= 3
      2840305.70     10267953.07      2840483.50     10267573.00
      2840255.67     10267403.10
#Sta/Elev= 30
  4580.4 1048.78  4617.1 1046.56  4663.1 1043.05  4685.9 1039.90  4691.4 1040.28
  4805.6 1034.41  4822.9 1029.91  4828.5 1029.96  4834.3 1028.75  4874.1 1029.05
  4971.0 1027.97  4988.3 1024.19  5020.4 1023.31  5020.5 1022.51  5021.0 1019.51
  5032.4 1019.51  5032.9 1022.51  5055.9 1022.89  5062.1 1025.06  5070.5 1025.83
  5076.7 1029.56  5091.3 1030.73  5097.6 1034.45  5103.0 1034.54  5112.2 1036.26
  5120.5 1035.80  5126.8 1036.91  5147.6 1037.58  5166.1 1037.14  5284.2 1038.07
#Mann=6,-1,0
  4580.4    0.12       0  4617.1    0.05       0  5020.5    0.05       0
  5032.9    0.05       0  5103.0    0.12       0  5166.1    0.05       0
Bank Sta=5020.5,5032.9
Exp/Cntr=0.3,0.1

Type RM Length L Ch R = 1,10176,478,478,478
BEGIN DESCRIPTION:
REED CREEK 21.0
END DESCRIPTION:
XS GIS Cut Line= 3
      2840855.68     10267803.11      2840924.50     10267503.00
      2840605.70     10267103.13
#Sta/Elev= 30
  4692.1 1038.43  4716.1 1038.56  4743.4 1036.88  4759.0 1035.26  4849.9 1032.09
  4887.0 1028.66  4892.8 1027.59  4897.9 1027.86  4935.7 1025.19  4969.1 1025.21
  4983.4 1022.12  4983.9 1019.12  4995.4 1019.12  4995.9 1022.12  5041.4 1022.99
  5055.8 1024.59  5063.8 1027.09  5070.2 1029.84  5076.6 1029.72  5091.1 1033.91
  5099.1 1034.75  5127.7 1034.25  5155.1 1035.16  5177.5 1035.17  5255.6 1034.20
  5383.5 1034.93  5447.5 1036.90  5454.6 1037.80  5489.8 1039.17  5511.4 1041.85
#Mann=3,-1,0
  4692.1    0.05       0  4983.4    0.05       0  4995.9    0.05       0
Bank Sta=4983.4,4995.9
Exp/Cntr=0.3,0.1

Type RM Length L Ch R = 1,9698,474,474,474
BEGIN DESCRIPTION:
REED CREEK 20.0
END DESCRIPTION:
XS GIS Cut Line= 3
      2841605.69     10267803.12      2841393.25     10267417.00
      2841155.68     10266703.09
#Sta/Elev= 30
  4559.3 1038.69  4703.0 1033.43  4752.0 1031.21  4795.6 1025.89  4817.9 1025.46
  4833.2 1030.09  4898.8 1031.04  4913.1 1030.01  4932.7 1025.81  4942.4 1021.87
  4948.1 1020.92  4958.5 1019.85  4970.2 1020.57  4974.0 1019.36  4974.5 1016.36
  4986.0 1016.36  4986.5 1019.36  4993.0 1020.42  5035.1 1021.51  5056.8 1023.61
  5072.0 1025.87  5098.4 1032.04  5204.3 1031.95  5319.9 1029.98  5436.2 1030.97
  5515.0 1033.46  5641.6 1039.47  5704.9 1044.57  5710.2 1045.99  5752.4 1047.97
#Mann=6,-1,0
  4559.3    0.12       0  4703.0    0.05       0  4817.9    0.12       0
  4932.7    0.05       0  4974.0    0.05       0  4986.5    0.05       0
Bank Sta=4974,4986.5
Exp/Cntr=0.3,0.1

Type RM Length L Ch R = 1,9224,431,431,431
BEGIN DESCRIPTION:
REED CREEK 19.0
END DESCRIPTION:
XS GIS Cut Line= 3
      2842155.68     10267353.11      2841806.50     10267215.00
      2841605.72     10267153.12
#Sta/Elev= 30
  4624.5 1057.28  4646.0 1055.01  4698.8 1045.03  4710.5 1043.72  4717.8 1041.84
  4742.1 1038.85  4747.5 1039.03  4753.5 1037.53  4825.9 1032.04  4835.0 1031.98
  4855.6 1029.59  4861.1 1028.08  4871.8 1028.62  4925.6 1025.24  4963.8 1020.70
  4979.4 1017.40  4982.6 1017.28  5005.0 1016.15  5005.5 1013.15  5017.2 1013.15
  5017.7 1016.15  5020.0 1017.38  5025.2 1018.54  5052.6 1020.50  5068.7 1023.34
  5080.1 1025.53  5090.5 1027.24  5095.8 1029.37  5105.5 1030.70  5210.1 1031.26
#Mann=8,-1,0
  4624.5    0.12       0  4698.8    0.05       0  4835.0    0.12       0
  4982.6    0.05       0  5005.0    0.05       0  5017.7    0.05       0
  5068.7    0.12       0  5080.1    0.05       0
Bank Sta=5005,5017.7
Exp/Cntr=0.3,0.1

Type RM Length L Ch R = 1,8793,1011,1011,1011
BEGIN DESCRIPTION:
Mapping XS 6f2454f5
END DESCRIPTION:
XS GIS Cut Line= 3
      2842445.94     10267381.48      2841980.27     10266750.58
      2841244.21     10266480.19
#Sta/Elev= 30
  4376.1 1044.81  4438.9 1048.08  4447.4 1046.98  4494.6 1048.23  4553.8 1048.38
  4566.6 1046.62  4603.9 1046.05  4618.6 1044.18  4624.8 1045.79  4657.8 1045.41
  4683.3 1045.08  4725.0 1041.55  4768.9 1035.33  4854.5 1026.48  4961.0 1020.31
  4975.6 1018.31  4990.1 1014.06  4990.6 1011.06  5002.3 1011.06  5002.8 1014.06
  5011.1 1015.86  5030.0 1016.22  5055.0 1020.96  5075.8 1028.22  5090.5 1030.09
  5168.9 1028.21  5457.8 1027.65  5655.1 1032.05  5807.5 1038.36  5944.4 1042.05
#Mann=7,-1,0
  4376.1    0.05       0  4494.6    0.12       0  4566.6    0.05       0
  4657.8    0.12       0  4990.1    0.07       0  5002.8    0.12       0
  5030.0    0.05       0
Bank Sta=4990.1,5002.8
Exp/Cntr=0.3,0.1

Type RM Length L Ch R = 1,7782,495,495,495
BEGIN DESCRIPTION:
REED CREEK 16.0
END DESCRIPTION:
XS GIS Cut Line= 3
      2842555.71     10266053.13      2842344.50     10265927.00
      2842005.64     10265803.10
#Sta/Elev= 30
  4754.0 1044.06  4756.9 1044.06  4767.6 1040.40  4777.3 1038.72  4789.0 1034.94
  4803.9 1033.05  4878.6 1023.11  4900.0 1021.49  4905.8 1021.73  4915.5 1019.99
  4921.4 1019.83  4928.7 1017.59  4936.9 1016.23  4952.0 1015.36  4958.3 1013.69
  4980.5 1010.97  4981.0 1007.97  4993.0 1007.97  4993.5 1010.97  5009.4 1011.02
  5020.0 1012.50  5025.6 1014.41  5041.3 1016.01  5062.6 1016.43  5081.4 1015.34
  5126.5 1021.64  5172.9 1023.82  5234.0 1027.38  5337.2 1030.98  5360.8 1032.24
#Mann=6,-1,0
  4754.0    0.12       0  4803.9    0.05       0  4980.5    0.03       0
  4993.5    0.05       0  5172.9    0.12       0  5337.2    0.05       0
Bank Sta=4980.5,4993.5
Exp/Cntr=0.3,0.1
