--- SANDY CREEK.prj (project) ---

Proj Title=SANDY CREEK Base Level Engineering
Current Plan=p01
Default Exp/Contr=0.3,0.1
English Units
Geom File=g01
Flow File=f01
Plan File=p01
BEGIN DESCRIPTION:
SANDY CREEK
END DESCRIPTION:

--- SANDY CREEK.p01 (plan) ---

Plan Title=Multiple Run
Short Identifier=Multiple
Geom File=g01
Flow File=f01
Subcritical Flow
K Sum by GR= 0
Std Step Tol= 0.01
Critical Tol= 0.01
Num of Std Step Trials= 20
Max Error Tol= 0.3
Flow Tol Ratio= 0.001
Split Flow NTrial= 30
Split Flow Tol= 0.02
Split Flow Ratio= 0.02
Log Output Level= 0
Friction Slope Method= 1
Unsteady Friction Slope Method= 2
Unsteady Bridges Friction Slope Method= 1
Parabolic Critical Depth
Global Vel Dist=  1 , 1 , 1
Global Log Level= 0
CheckData=True
Encroach Param= -1, 0, 0, 0
BEGIN DESCRIPTION:
Multiple Run
END DESCRIPTION:

--- SANDY CREEK.f01 (steady flow) ---

Flow Title=Multiple
Number of Profiles=7
Profile Names=10-year,25-year,50-year,1pct_min,100-year,1pct_plu,500-year
River Rch & RM= SANDY CREEK,Reach-1,29298
      71     138     216     113     340    1026     901
River Rch & RM= SANDY CREEK,Reach-1,18739
      74     147     231     121     365    1103     974
River Rch & RM= SANDY CREEK,Reach-1,15365
     166     358     589     319     964    2910    2739
River Rch & RM= SANDY CREEK,Reach-1,11029
     197     432     717     390    1179    3561    3391
River Rch & RM= SANDY CREEK,Reach-1,6797
     244     543     909     499    1506    4548    4389
Boundary for River Rch & Prof#=SANDY CREEK,Reach-1,1
Up Type=0
Dn Type=3
Dn Slope=0.005
Boundary for River Rch & Prof#=SANDY CREEK,Reach-1,2
Up Type=0
Dn Type=3
Dn Slope=0.005
Boundary for River Rch & Prof#=SANDY CREEK,Reach-1,3
Up Type=0
Dn Type=3
Dn Slope=0.005
Boundary for River Rch & Prof#=SANDY CREEK,Reach-1,4
Up Type=0
Dn Type=3
Dn Slope=0.005
Boundary for River Rch & Prof#=SANDY CREEK,Reach-1,5
Up Type=0
Dn Type=3
Dn Slope=0.005
Boundary for River Rch & Prof#=SANDY CREEK,Reach-1,6
Up Type=0
Dn Type=3
Dn Slope=0.005
Boundary for River Rch & Prof#=SANDY CREEK,Reach-1,7
Up Type=0
Dn Type=3
Dn Slope=0.005

--- SANDY CREEK.g01 (geometry) ---

Geom Title=Existing Conditions

River Reach=SANDY CREEK,Reach-1
Reach XY= 30
      2874979.75     10251630.00      2875413.00     10250792.00
      2875408.50     10250405.00      2875140.25     10250114.00
      2875274.25     10249615.00      2875565.75     10249444.00
      2875955.50     10248617.00      2876100.00     10247774.00
      2876580.75     10247621.00      2876526.00     10247129.00
      2877006.00     10246691.00      2876941.75     10244513.00
      2877238.50     10244322.00      2877199.75     10243345.00
      2877482.25     10242854.00      2876891.25     10241116.00
      2877254.25     10239807.00      2876966.75     10239479.00
      2876901.25     10238798.00      2876374.00     10238158.00
      2876817.00     10235099.00      2876215.50     10233965.00
      2875013.00     10233630.00      2874081.75     10232260.00
      2873868.25     10231392.00      2873399.25     10231068.00
      2873584.75     10230579.00      2874619.25     10229848.00
      2874698.00     10228678.00      2875195.25     10227729.00

Type RM Length L Ch R = 1,29298,363,363,363
BEGIN DESCRIPTION:
SANDY CREEK 58.0
END DESCRIPTION:
XS GIS Cut Line= 3
      2875355.70     10251553.14      2875171.50     10251275.00
      2874905.70     10251253.11
#Sta/Elev= 30
  4666.4 1095.77  4674.0 1095.50  4680.0 1095.78  4716.1 1093.65  4725.1 1093.70
  4731.1 1093.14  4761.2 1091.91  4767.2 1092.35  4774.4 1092.37  4782.3 1091.09
  4797.3 1090.74  4846.3 1088.48  4875.5 1088.12  4882.3 1087.79  4890.6 1088.02
  4896.6 1087.31  4962.8 1085.67  4998.0 1083.88  4998.3 1080.88  5001.8 1080.88
  5002.0 1083.88  5035.9 1086.14  5046.0 1086.41  5082.5 1089.21  5146.3 1092.07
  5156.3 1092.88  5186.4 1094.33  5246.6 1097.87  5256.7 1098.76  5266.7 1099.00
#Mann=3,-1,0
  4666.4    0.05       0  4998.0    0.03       0  5002.0    0.05       0
Bank Sta=4998,5002
Exp/Cntr=0.3,0.1

Type RM Length L Ch R = 1,28935,389,389,389
BEGIN DESCRIPTION:
SANDY CREEK 57.0
END DESCRIPTION:
XS GIS Cut Line= 3
      2875855.71     10251153.12      2875311.75     10250951.00
      2875005.64     10251053.13
#Sta/Elev= 30
  4419.7 1093.97  4459.9 1092.19  4465.3 1092.92  4490.3 1090.71  4515.3 1090.15
  4520.6 1090.59  4537.1 1089.44  4545.7 1089.34  4551.0 1090.78  4576.0 1088.24
  4596.7 1087.47  4606.4 1087.60  4654.4 1085.30  4686.4 1084.94  4692.1 1084.22
  4717.1 1084.25  4785.6 1081.64  4808.2 1080.28  4814.4 1081.49  4833.2 1082.09
  4942.5 1081.70  4979.7 1080.69  4985.1 1079.70  4993.2 1079.60  4993.5 1076.60
  4997.0 1076.60  4997.2 1079.60  5085.6 1083.60  5132.9 1084.68  5322.7 1091.60
#Mann=5,-1,0
  4419.7    0.05       0  4596.7    0.12       0  4785.6    0.05       0
  4993.2    0.03       0  4997.2    0.05       0
Bank Sta=4993.2,4997.2
Exp/Cntr=0.3,0.1

Type RM Length L Ch R = 1,28546,48,48,48
BEGIN DESCRIPTION:
Mapping XS eef3483a
END DESCRIPTION:
XS GIS Cut Line= 4
      2875823.90     10250894.66      2875539.80     10250714.22
      2875424.64     10250648.96      2875114.26     10250798.40
#Sta/Elev= 30
  4532.4 1089.81  4576.8 1089.19  4582.8 1089.85  4603.9 1088.79  4657.0 1088.76
  4676.8 1089.23  4707.3 1088.70  4713.2 1089.26  4728.4 1088.56  4770.9 1088.48
  4779.1 1087.64  4807.2 1087.34  4858.9 1084.54  4864.8 1084.73  4868.4 1083.98
  4886.1 1083.38  4923.7 1080.73  4954.1 1074.88  4980.8 1071.87  4981.1 1068.87
  4984.6 1068.87  4984.8 1071.87  4997.8 1072.30  5019.6 1071.89  5042.2 1073.66
  5070.4 1076.93  5160.9 1079.96  5222.1 1083.41  5288.7 1085.88  5345.8 1086.98
#Mann=5,-1,0
  4532.4    0.05       0  4657.0    0.12       0  4770.9    0.05       0
  4980.8    0.05       0  4984.8    0.05       0
Bank Sta=4980.8,4984.8
Exp/Cntr=0.3,0.1

Type RM Length L Ch R = 1,28498,62,62,62
BEGIN DESCRIPTION:
Mapping XS 328af43f
END DESCRIPTION:
XS GIS Cut Line= 6
      2875839.25     10250810.20      2875493.74     10250645.12
      2875474.54     10250610.57      2875436.16     10250599.06
      2875355.54     10250618.25      2875105.99     10250737.27
#Sta/Elev= 30
  4516.7 1090.15  4614.6 1090.70  4710.9 1089.64  4778.9 1086.77  4786.6 1087.35
  4841.4 1083.04  4864.1 1082.60  4902.8 1079.92  4906.8 1078.10  4922.8 1080.16
  4928.5 1078.87  4934.8 1080.79  4941.2 1080.79  4945.4 1079.38  4950.7 1081.42
  4976.9 1077.73  4989.9 1077.22  5022.1 1078.35  5026.2 1080.00  5029.5 1076.49
  5029.7 1073.49  5033.2 1073.49  5033.5 1076.49  5051.6 1079.54  5073.1 1076.79
  5087.4 1076.71  5150.0 1078.66  5200.9 1081.86  5261.5 1084.08  5338.7 1085.00
#Mann=3,-1,0
  4516.7    0.05       0  5029.5    0.05       0  5033.5    0.05       0
Bank Sta=5029.5,5033.5
Exp/Cntr=0.3,0.1

Type RM Length L Ch R = 1,28436,421,421,421
BEGIN DESCRIPTION:
Mapping XS 29f7bdee
END DESCRIPTION:
XS GIS Cut Line= 4
      2875747.13     10250625.94      2875405.45     10250541.48
      2875140.58     10250583.70      2875064.98     10250659.30
#Sta/Elev= 30
  4643.6 1087.33  4665.7 1087.15  4686.3 1086.52  4706.9 1086.50  4727.5 1085.50
  4756.4 1085.05  4761.6 1084.25  4797.8 1083.12  4851.1 1080.42  4861.4 1080.20
  4880.7 1079.12  4885.9 1079.19  4927.3 1076.70  4968.7 1074.85  4974.7 1074.34
  4985.0 1072.74  4990.9 1072.36  4991.1 1069.36  4994.6 1069.36  4994.9 1072.36
  5025.7 1073.11  5046.0 1074.06  5066.2 1075.46  5157.3 1077.48  5238.4 1081.21
  5309.3 1082.35  5316.3 1082.83  5323.4 1082.55  5351.7 1083.25  5370.7 1083.30
#Mann=3,-1,0
  4643.6    0.05       0  4990.9    0.05       0  4994.9    0.05       0
Bank Sta=4990.9,4994.9
Exp/Cntr=0.3,0.1

Type RM Length L Ch R = 1,28015,484,484,484
BEGIN DESCRIPTION:
SANDY CREEK 55.0
END DESCRIPTION:
XS GIS Cut Line= 3
      2875505.66     10250253.11      2875188.50     10250248.00
      2875105.68     10250453.11
#Sta/Elev= 30
  4682.8 1077.81  4742.8 1075.40  4782.8 1074.16  4802.8 1074.02  4832.8 1073.37
  4862.8 1072.54  4872.8 1071.99  4892.8 1071.68  4932.8 1070.41  4972.8 1068.52
  4982.8 1067.79  4993.4 1067.53  4993.7 1064.53  4997.2 1064.53  4997.4 1067.53
  5005.5 1069.23  5050.8 1070.98  5069.6 1072.15  5075.0 1072.20  5091.8 1073.08
  5099.1 1073.81  5104.5 1073.43  5123.2 1074.11  5134.9 1073.71  5152.8 1075.22
  5176.9 1076.07  5182.3 1076.05  5199.6 1077.14  5211.8 1077.31  5221.2 1077.86
#Mann=3,-1,0
  4682.8    0.05       0  4993.4    0.03       0  4997.4    0.05       0
Bank Sta=4993.4,4997.4
Exp/Cntr=0.3,0.1

Type RM Length L Ch R = 1,27531,459,459,459
BEGIN DESCRIPTION:
SANDY CREEK 54.0
END DESCRIPTION:
XS GIS Cut Line= 3
      2875455.70     10250003.12      2875237.00     10249821.00
      2875055.66     10249703.10
#Sta/Elev= 30
  4715.4 1073.53  4751.2 1072.00  4786.4 1070.01  4871.6 1068.08  4936.1 1065.51
  4949.7 1064.33  4963.4 1062.47  4971.2 1062.40  4985.5 1063.26  4997.6 1062.20
  5002.6 1062.20  5004.4 1061.26  5004.7 1058.26  5008.2 1058.26  5008.4 1061.26
  5013.5 1061.54  5021.6 1063.39  5027.5 1063.80  5049.3 1063.87  5072.9 1064.92
  5078.9 1064.94  5094.0 1066.47  5108.9 1066.47  5121.1 1066.98  5144.7 1068.40
  5157.3 1069.60  5180.5 1071.08  5208.7 1072.34  5213.3 1073.15  5216.3 1073.15
#Mann=3,-1,0
  4715.4    0.05       0  5004.4    0.05       0  5008.4    0.05       0
Bank Sta=5004.4,5008.4
Exp/Cntr=0.3,0.1

Type RM Length L Ch R = 1,27072,305,305,305
BEGIN DESCRIPTION:
SANDY CREEK 53.0
END DESCRIPTION:
XS GIS Cut Line= 3
      2875705.66     10249753.08      2875433.25     10249484.00
      2875205.64     10249453.11
#Sta/Elev= 30
  4617.1 1074.75  4620.6 1074.75  4624.1 1073.95  4673.6 1072.14  4687.7 1070.96
  4716.0 1069.77  4758.4 1067.19  4808.0 1065.19  4829.2 1063.76  4907.0 1060.56
  4921.1 1059.11  4928.2 1057.80  4935.3 1057.70  4942.3 1059.11  4956.4 1059.48
  4963.6 1059.25  4982.7 1056.35  4983.0 1053.35  4986.5 1053.35  4986.7 1056.35
  4997.1 1056.71  5043.4 1056.72  5048.4 1058.17  5058.1 1059.36  5068.2 1061.14
  5088.4 1061.62  5115.9 1063.53  5120.9 1063.51  5199.4 1067.88  5229.7 1069.11
#Mann=3,-1,0
  4617.1    0.05       0  4982.7    0.05       0  4986.7    0.05       0
Bank Sta=4982.7,4986.7
Exp/Cntr=0.3,0.1

Type RM Length L Ch R = 1,26767,38,38,38
BEGIN DESCRIPTION:
Mapping XS 23d10475
END DESCRIPTION:
XS GIS Cut Line= 4
      2875869.96     10249512.73      2875620.41     10249324.61
      2875539.80     10249274.71      2875225.43     10249198.03
#Sta/Elev= 30
  4631.7 1067.48  4641.3 1066.99  4655.9 1067.92  4662.2 1067.44  4670.5 1067.86
  4712.2 1067.02  4720.4 1067.74  4726.7 1066.68  4785.0 1065.36  4826.6 1063.37
  4884.9 1058.94  4941.1 1057.78  4949.9 1057.20  4956.1 1055.45  4971.5 1052.91
  4990.7 1052.20  4991.0 1049.20  4994.5 1049.20  4994.7 1052.20  5008.1 1052.55
  5014.0 1053.88  5029.4 1053.79  5035.3 1055.34  5053.5 1055.90  5084.4 1058.65
  5104.5 1059.68  5249.1 1063.95  5276.4 1063.95  5359.7 1066.46  5362.6 1067.03
#Mann=3,-1,0
  4631.7    0.05       0  4990.7    0.05       0  4994.7    0.05       0
Bank Sta=4990.7,4994.7
Exp/Cntr=0.3,0.1

Type RM Length L Ch R = 1,26729,182,182,182
BEGIN DESCRIPTION:
Mapping XS 1503cd76
END DESCRIPTION:
XS GIS Cut Line= 6
      2875881.46     10249497.38      2875735.57     10249309.26
      2875628.09     10249282.39      2875585.87     10249259.35
      2875528.29     10249255.52      2875274.94     10249128.85
#Sta/Elev= 30
  4608.2 1065.84  4693.5 1065.94  4722.4 1064.60  4778.5 1063.86  4828.7 1061.23
  4848.6 1061.21  4851.1 1060.24  4866.8 1059.48  4931.6 1057.52  4931.9 1054.52
  4935.4 1054.52  4935.6 1057.52  4955.7 1060.64  4961.3 1060.64  4965.7 1058.52
  4971.4 1060.61  5007.7 1060.90  5022.1 1060.00  5027.1 1061.13  5035.4 1061.19
  5055.4 1060.26  5075.4 1058.19  5081.0 1058.73  5088.1 1057.93  5103.3 1058.14
  5215.1 1062.23  5231.9 1063.68  5237.5 1063.15  5254.3 1063.84  5346.1 1068.32
#Mann=3,-1,0
  4608.2    0.05       0  4931.6    0.05       0  4935.6    0.05       0
Bank Sta=4931.6,4935.6
Exp/Cntr=0.3,0.1

Type RM Length L Ch R = 1,26547,383,383,383
BEGIN DESCRIPTION:
Mapping XS 6309e039
END DESCRIPTION:
XS GIS Cut Line= 6
      2875916.00     10249581.84      2875892.96     10249355.32
      2875789.32     10249240.16      2875593.54     10249117.32
      2875516.77     10249071.26      2875069.15     10248975.61
#Sta/Elev= 30
  4377.7 1067.88  4476.9 1064.88  4525.6 1064.40  4587.5 1062.39  4654.5 1061.87
  4819.2 1057.67  4847.2 1056.00  4855.7 1056.34  4861.6 1055.31  4870.9 1055.56
  4876.9 1054.09  4913.4 1054.55  4919.3 1053.40  4928.7 1054.37  4934.7 1053.09
  4986.5 1053.15  4988.7 1051.62  4988.9 1048.62  4992.4 1048.62  4992.7 1051.62
  5013.7 1051.91  5035.6 1057.27  5084.1 1059.74  5102.5 1061.51  5184.3 1064.77
  5339.1 1073.61  5378.3 1074.92  5383.5 1074.33  5460.4 1074.43  5538.7 1075.29
#Mann=3,-1,0
  4377.7    0.05       0  4988.7    0.05       0  4992.7    0.05       0
Bank Sta=4988.7,4992.7
Exp/Cntr=0.3,0.1

Type RM Length L Ch R = 1,26164,480,480,480
BEGIN DESCRIPTION:
SANDY CREEK 51.0
END DESCRIPTION:
XS GIS Cut Line= 3
      2875955.67     10249353.07      2875818.25     10248861.00
      2875555.67     10248853.11
#Sta/Elev= 30
  4489.1 1060.82  4506.1 1059.88  4511.3 1060.31  4530.6 1059.61  4545.5 1059.85
  4551.4 1059.36  4619.0 1057.97  4800.2 1055.68  4831.7 1054.12  4852.5 1053.82
  4913.1 1051.26  4918.3 1051.57  4952.4 1051.12  4966.7 1051.58  4986.6 1049.09
  4989.8 1048.33  4990.0 1045.33  4993.5 1045.33  4993.8 1048.33  4996.3 1048.98
  5012.6 1049.57  5042.6 1049.77  5072.6 1051.55  5096.9 1052.13  5182.6 1058.21
  5192.7 1058.41  5222.7 1060.88  5252.7 1062.17  5260.2 1063.74  5262.7 1063.74
#Mann=3,-1,0
  4489.1    0.05       0  4989.8    0.05       0  4993.8    0.05       0
Bank Sta=4989.8,4993.8
Exp/Cntr=0.3,0.1

Type RM Length L Ch R = 1,25684,457,457,457
BEGIN DESCRIPTION:
SANDY CREEK 50.0
END DESCRIPTION:
XS GIS Cut Line= 3
      2876305.66     10248753.08      2876010.00     10248463.00
      2875755.69     10248303.11
#Sta/Elev= 30
  4585.8 1052.25  4589.3 1052.25  4592.8 1049.06  4599.8 1048.85  4607.0 1046.26
  4628.1 1044.08  4635.3 1045.91  4649.4 1046.41  4727.1 1044.90  4776.7 1047.97
  4840.3 1048.32  4974.7 1044.83  4995.9 1043.45  4999.5 1041.91  5008.1 1041.59
  5008.3 1038.59  5011.8 1038.59  5012.1 1041.59  5025.4 1043.41  5061.9 1043.80
  5067.8 1042.55  5089.0 1044.64  5125.5 1045.46  5134.9 1046.67  5140.8 1046.13
  5198.5 1050.77  5271.5 1054.72  5292.8 1055.09  5297.4 1056.79  5300.4 1056.79
#Mann=3,-1,0
  4585.8    0.05       0  5008.1    0.05       0  5012.1    0.05       0
Bank Sta=5008.1,5012.1
Exp/Cntr=0.3,0.1

Type RM Length L Ch R = 1,25227,451,451,451
BEGIN DESCRIPTION:
SANDY CREEK 49.0
END DESCRIPTION:
XS GIS Cut Line= 3
      2876405.70     10248203.12      2876146.75     10248081.00
      2876005.68     10248053.11
#Sta/Elev= 30
  4713.7 1052.12  4721.4 1051.83  4780.1 1047.50  4790.7 1047.07  4813.2 1045.33
  4824.5 1043.97  4864.5 1041.41  4870.1 1041.71  4887.3 1040.32  4910.1 1041.24
  4915.6 1040.44  4932.9 1040.79  4938.4 1039.97  4961.2 1039.66  4978.4 1037.84
  4984.0 1037.95  4990.1 1036.80  4995.8 1035.06  4996.1 1032.06  4999.6 1032.06
  4999.8 1035.06  5010.5 1035.91  5021.5 1038.03  5031.7 1039.04  5041.9 1039.45
  5052.1 1040.70  5066.9 1040.63  5072.4 1041.34  5133.6 1044.90  5143.8 1046.04
#Mann=4,-1,0
  4713.7    0.12       0  4721.4    0.05       0  4995.8    0.05       0
  4999.8    0.05       0
Bank Sta=4995.8,4999.8
Exp/Cntr=0.3,0.1

Type RM Length L Ch R = 1,24776,480,480,480
BEGIN DESCRIPTION:
SANDY CREEK 48.0
END DESCRIPTION:
XS GIS Cut Line= 3
      2876505.69     10248053.11      2876194.25     10247752.00
      2876155.70     10247653.15
#Sta/Elev= 30
  4566.8 1051.10  4588.0 1048.47  4624.6 1046.67  4644.6 1045.19  4651.6 1045.42
  4658.8 1044.53  4665.7 1044.54  4679.9 1042.49  4701.9 1040.86  4736.5 1038.66
  4750.6 1038.81  4778.9 1037.70  4849.6 1037.44  4892.1 1038.19  4927.6 1037.71
  4955.9 1036.04  4962.8 1034.62  4975.0 1033.52  4975.2 1030.52  4978.7 1030.52
  4979.0 1033.52  5002.1 1033.95  5007.0 1035.59  5012.4 1034.99  5020.3 1038.03
  5042.2 1040.97  5061.4 1042.30  5066.7 1042.06  5091.2 1044.19  5106.1 1044.31
#Mann=5,-1,0
  4566.8    0.05       0  4624.6    0.12       0  4701.9    0.05       0
  4975.0    0.05       0  4979.0    0.05       0
Bank Sta=4975,4979
Exp/Cntr=0.3,0.1

Type RM Length L Ch R = 1,24296,482,482,482
BEGIN DESCRIPTION:
SANDY CREEK 47.0
END DESCRIPTION:
XS GIS Cut Line= 3
      2876655.64     10247553.14      2876598.75     10247592.00
      2876305.72     10247553.12
#Sta/Elev= 30
  4931.1 1041.29  4934.1 1041.29  4938.5 1040.03  4953.4 1037.93  4959.5 1038.15
  4967.4 1036.32  4974.4 1031.79  4980.5 1032.20  4989.3 1029.94  4993.4 1029.67
  4993.6 1026.67  4997.1 1026.67  4997.4 1029.67  4998.8 1030.24  5004.1 1030.24
  5013.2 1031.30  5028.9 1031.77  5063.6 1032.42  5083.8 1032.24  5107.3 1032.77
  5134.2 1034.02  5174.6 1034.94  5180.6 1035.62  5185.7 1035.59  5204.8 1037.35
  5245.2 1039.42  5253.9 1039.63  5259.0 1039.36  5265.4 1039.78  5295.6 1040.63
#Mann=3,-1,0
  4931.1    0.05       0  4993.4    0.05       0  4997.4    0.05       0
Bank Sta=4993.4,4997.4
Exp/Cntr=0.3,0.1

Type RM Length L Ch R = 1,23814,470,470,470
BEGIN DESCRIPTION:
SANDY CREEK 46.0
END DESCRIPTION:
XS GIS Cut Line= 3
      2876805.68     10247453.11      2876526.00     10247129.00
      2876355.72     10247203.09
#Sta/Elev= 30
  4571.9 1041.30  4650.3 1036.47  4658.5 1036.50  4742.5 1031.67  4820.4 1029.02
  4841.2 1029.13  4848.9 1028.40  4884.0 1027.77  4919.1 1028.70  4926.8 1028.13
  4933.4 1028.92  4947.6 1028.08  4961.9 1028.50  4976.1 1027.74  4982.7 1025.67
  4990.4 1026.04  4994.4 1024.99  4994.7 1021.99  4998.2 1021.99  4998.4 1024.99
  5019.8 1027.09  5033.1 1027.17  5048.7 1029.23  5054.9 1029.16  5095.5 1033.27
  5131.2 1033.97  5142.1 1034.43  5147.9 1035.55  5153.3 1034.99  5185.7 1036.39
#Mann=4,-1,0
  4571.9    0.12       0  4658.5    0.05       0  4994.4    0.05       0
  4998.4    0.05       0
Bank Sta=4994.4,4998.4
Exp/Cntr=0.3,0.1

Type RM Length L Ch R = 1,23344,482,482,482
BEGIN DESCRIPTION:
SANDY CREEK 45.0
END DESCRIPTION:
XS GIS Cut Line= 3
      2877105.73     10246953.12      2876916.50     10246936.00
      2876405.70     10246803.12
#Sta/Elev= 30
  4810.0 1032.15  4850.2 1029.77  4865.4 1028.35  4920.5 1025.32  4950.6 1024.24
  4960.7 1024.40  4970.7 1022.58  4974.1 1020.60  4974.4 1017.60  4977.9 1017.60
  4978.1 1020.60  5029.0 1021.14  5052.5 1023.88  5069.5 1024.95  5074.7 1024.63
  5110.1 1025.46  5185.9 1026.11  5191.1 1025.75  5207.5 1026.39  5272.2 1026.96
  5290.2 1027.98  5312.7 1027.98  5362.5 1029.18  5383.2 1029.82  5388.6 1030.74
  5403.8 1030.48  5414.2 1031.26  5429.1 1031.49  5505.0 1035.53  5527.8 1036.09
#Mann=3,-1,0
  4810.0    0.05       0  4974.1    0.05       0  4978.1    0.05       0
Bank Sta=4974.1,4978.1
Exp/Cntr=0.3,0.1

Type RM Length L Ch R = 1,22862,468,468,468
BEGIN DESCRIPTION:
SANDY CREEK 44.0
END DESCRIPTION:
XS GIS Cut Line= 3
      2877155.72     10246503.12      2876996.75     10246473.00
      2876755.71     10246553.10
#Sta/Elev= 30
  4838.2 1025.83  4858.6 1025.19  4878.9 1023.37  4909.5 1021.63  4940.0 1018.98
  4960.4 1018.84  4969.0 1017.32  4974.1 1017.51  4980.7 1015.55  5003.2 1015.17
  5014.6 1013.68  5014.8 1010.68  5018.3 1010.68  5018.6 1013.68  5022.2 1016.68
  5032.7 1020.55  5043.0 1021.40  5048.2 1021.14  5053.8 1021.71  5074.6 1020.75
  5085.4 1021.24  5111.6 1021.01  5117.0 1021.58  5137.9 1021.68  5148.7 1022.26
  5159.2 1022.00  5222.4 1024.01  5232.9 1024.72  5238.2 1024.03  5254.0 1024.55
#Mann=3,-1,0
  4838.2    0.05       0  5014.6    0.05       0  5018.6    0.05       0
Bank Sta=5014.6,5018.6
Exp/Cntr=0.3,0.1

Type RM Length L Ch R = 1,22394,663,663,663
BEGIN DESCRIPTION:
SANDY CREEK 43.0
END DESCRIPTION:
XS GIS Cut Line= 3
      2877255.67     10246203.10      2877035.75     10246039.00
      2876455.67     10245953.11
#Sta/Elev= 30
  4725.6 1025.86  4833.0 1020.73  4853.8 1020.35  4939.3 1016.49  4947.6 1015.34
  4953.9 1015.35  4975.1 1013.43  5002.6 1013.20  5003.6 1011.55  5003.8 1008.55
  5007.3 1008.55  5007.6 1011.55  5010.6 1012.90  5020.3 1013.17  5030.4 1014.47
  5040.5 1017.12  5050.6 1017.43  5080.9 1016.58  5161.8 1015.98  5252.8 1017.12
  5313.4 1015.70  5323.6 1016.16  5333.7 1018.07  5364.0 1018.36  5417.6 1021.15
  5465.1 1022.79  5482.1 1022.67  5515.6 1024.25  5551.6 1027.18  5586.4 1027.72
#Mann=3,-1,0
  4725.6    0.05       0  5003.6    0.05       0  5007.6    0.05       0
Bank Sta=5003.6,5007.6
Exp/Cntr=0.3,0.1

Type RM Length L Ch R = 1,21731,197,197,197
BEGIN DESCRIPTION:
Mapping XS 531fbbfe
END DESCRIPTION:
XS GIS Cut Line= 2
      2877638.99     10245416.33      2876119.37     10245478.78
#Sta/Elev= 30
  4248.2 1017.78  4351.6 1014.88  4751.9 1015.54  4922.1 1011.95  4984.2 1007.14
  5000.1 1005.15  5000.4 1002.15  5003.9 1002.15  5004.1 1005.15  5012.1 1006.83
  5017.4 1010.02  5019.7 1011.41  5024.7 1007.89  5032.2 1010.98  5042.2 1012.00
  5092.2 1012.20  5172.3 1010.97  5192.3 1011.78  5222.3 1009.78  5242.3 1014.00
  5272.4 1015.72  5332.4 1015.99  5382.5 1013.06  5402.5 1013.43  5422.5 1016.69
  5513.4 1020.43  5582.6 1019.08  5662.7 1019.75  5692.7 1018.08  5769.1 1021.71
#Mann=5,-1,0
  4248.2    0.05       0  4984.2    0.12       0  5000.1    0.07       0
  5004.1    0.12       0  5017.4    0.05       0
Bank Sta=5000.1,5004.1
Exp/Cntr=0.3,0.1

Type RM Length L Ch R = 1,21534,138,138,138
BEGIN DESCRIPTION:
Mapping XS fe558d50
END DESCRIPTION:
XS GIS Cut Line= 3
      2877681.82     10245336.22      2876906.37     10245278.63
      2876078.95     10245228.83
#Sta/Elev= 30
  4296.0 1017.00  4392.4 1016.70  4522.8 1014.74  4544.1 1015.49  4814.6 1015.14
  4974.0 1011.21  5002.1 1005.35  5002.3 1002.35  5005.8 1002.35  5006.1 1005.35
  5064.2 1010.61  5184.5 1010.84  5204.5 1010.18  5214.5 1008.35  5244.1 1009.50
  5254.6 1008.06  5364.8 1015.03  5404.9 1015.94  5412.5 1014.62  5417.5 1015.82
  5455.0 1012.62  5465.0 1012.76  5495.0 1014.76  5555.1 1014.53  5575.2 1015.88
  5595.2 1015.27  5605.2 1016.57  5675.4 1016.84  5825.6 1023.05  5902.5 1024.80
#Mann=3,-1,0
  4296.0    0.05       0  5002.1    0.03       0  5006.1    0.05       0
Bank Sta=5002.1,5006.1
Exp/Cntr=0.3,0.1

Type RM Length L Ch R = 1,21396,441,441,441
BEGIN DESCRIPTION:
Mapping XS 8c5d00aa
END DESCRIPTION:
XS GIS Cut Line= 2
      2877597.24     10245187.16      2876201.43     10245103.83
#Sta/Elev= 30
  4369.5 1015.91  4401.1 1016.18  4471.2 1014.92  4541.4 1015.20  4561.4 1016.17
  4571.4 1014.96  4761.8 1014.46  4862.0 1012.69  4942.1 1010.21  4962.1 1007.72
  4982.1 1006.17  4992.2 1006.26  5000.2 1004.95  5000.4 1001.95  5003.9 1001.95
  5004.2 1004.95  5021.0 1008.33  5042.3 1009.28  5092.3 1008.74  5190.0 1009.38
  5232.6 1007.18  5252.6 1010.04  5262.6 1013.13  5302.7 1016.06  5422.9 1019.57
  5523.1 1020.13  5563.2 1022.46  5633.3 1022.27  5692.2 1018.79  5767.8 1019.79
#Mann=3,-1,0
  4369.5    0.05       0  5000.2    0.05       0  5004.2    0.05       0
Bank Sta=5000.2,5004.2
Exp/Cntr=0.3,0.1

Type RM Length L Ch R = 1,20955,449,449,449
BEGIN DESCRIPTION:
SANDY CREEK 40.0
END DESCRIPTION:
XS GIS Cut Line= 3
      2877255.71     10245003.14      2877011.25     10244723.00
      2876755.71     10244803.10
#Sta/Elev= 30
  4628.2 1013.42  4699.0 1011.78  4706.6 1012.03  4713.2 1011.38  4755.9 1010.39
  4905.0 1008.11  4925.8 1007.29  4933.4 1007.65  4940.1 1006.41  4954.3 1006.65
  4961.0 1004.91  4968.6 1005.83  4975.2 1003.55  4982.8 1004.26  4987.4 1002.78
  4987.7  999.78  4991.2  999.78  4991.4 1002.78  5005.8 1003.68  5037.3 1003.82
  5046.5 1004.92  5079.0 1006.57  5142.1 1006.53  5173.5 1009.09  5186.7 1009.27
  5194.5 1010.38  5213.9 1011.64  5219.2 1011.46  5257.3 1014.77  5267.8 1014.82
#Mann=3,-1,0
  4628.2    0.05       0  4987.4    0.05       0  4991.4    0.05       0
Bank Sta=4987.4,4991.4
Exp/Cntr=0.3,0.1

Type RM Length L Ch R = 1,20506,483,483,483
BEGIN DESCRIPTION:
SANDY CREEK 39.0
END DESCRIPTION:
XS GIS Cut Line= 3
      2877455.67     10244803.09      2877094.75     10244382.00
      2876555.72     10244103.13
#Sta/Elev= 30
  4445.4 1013.12  4468.7 1012.92  4495.3 1012.61  4509.6 1013.17  4537.6 1012.06
  4551.3 1012.51  4584.4 1011.90  4729.9 1009.75  4787.1 1007.54  4921.4 1002.88
  4948.6 1003.84  4962.9 1002.82  4977.1 1003.02  4996.0 1000.45  5006.5 1000.75
  5010.1 1000.19  5010.4  997.19  5013.9  997.19  5014.1 1000.19  5034.3 1001.51
  5044.0 1002.98  5050.8 1004.83  5056.4 1005.30  5089.0 1005.56  5111.5 1004.15
  5178.0 1007.00  5235.4 1006.86  5294.3 1008.20  5471.8 1014.59  5606.9 1018.73
#Mann=8,-1,0
  4445.4    0.12       0  4468.7    0.05       0  4584.4    0.12       0
  4729.9    0.05       0  4787.1    0.12       0  4921.4    0.05       0
  5010.1    0.03       0  5014.1    0.05       0
Bank Sta=5010.1,5014.1
Exp/Cntr=0.3,0.1

Type RM Length L Ch R = 1,20023,425,425,425
BEGIN DESCRIPTION:
SANDY CREEK 38.0
END DESCRIPTION:
XS GIS Cut Line= 3
      2877405.69     10244253.12      2877163.00     10244016.00
      2876905.67     10243953.11
#Sta/Elev= 30
  4660.7 1007.73  4667.8 1007.18  4690.3 1006.98  4710.2 1007.45  4731.4 1006.54
  4823.4 1006.08  4851.7 1005.58  4865.8 1004.72  4872.8 1004.97  4880.0 1003.86
  4894.1 1002.96  4901.1 1003.06  4950.7 1000.42  4957.7 1001.08  4964.8  999.48
  4971.8  999.24  4977.0  997.19  4977.2  994.19  4980.7  994.19  4981.0  997.19
  4986.0  997.91  4998.5  997.63  5017.8  999.03  5038.4  998.33  5059.0 1001.17
  5074.9 1002.72  5110.5 1003.37  5121.7 1003.07  5205.0 1004.97  5264.9 1007.71
#Mann=4,-1,0
  4660.7    0.12       0  4690.3    0.05       0  4977.0    0.03       0
  4981.0    0.05       0
Bank Sta=4977,4981
Exp/Cntr=0.3,0.1

Type RM Length L Ch R = 1,19598,388,388,388
BEGIN DESCRIPTION:
SANDY CREEK 37.0
END DESCRIPTION:
XS GIS Cut Line= 3
      2877805.69     10243803.12      2877219.25     10243612.00
      2876905.72     10243503.12
#Sta/Elev= 30
  4383.2 1008.07  4393.7 1007.83  4399.2 1006.95  4431.1 1005.12  4461.4 1004.04
  4493.6 1002.83  4551.5 1000.84  4564.0  998.57  4572.5 1000.57  4590.6 1002.97
  4687.1 1003.58  4691.6 1003.10  4849.2 1002.20  4930.1 1001.11  4972.2  998.70
  4978.9  997.17  4984.1  997.34  4997.2  995.36  4997.5  992.36  5001.0  992.36
  5001.2  995.36  5024.9  996.48  5041.6  998.28  5067.3  998.42  5134.9 1001.09
  5197.2 1004.56  5215.5 1004.77  5228.3 1006.13  5279.0 1008.14  5331.9 1011.50
#Mann=7,-1,0
  4383.2    0.05       0  4461.4    0.12       0  4493.6    0.05       0
  4687.1    0.12       0  4849.2    0.05       0  4997.2    0.03       0
  5001.2    0.05       0
Bank Sta=4997.2,5001.2
Exp/Cntr=0.3,0.1

Type RM Length L Ch R = 1,19210,471,471,471
BEGIN DESCRIPTION:
SANDY CREEK 36.0
END DESCRIPTION:
XS GIS Cut Line= 3
      2877855.69     10243503.11      2877255.75     10243242.00
      2877105.66     10243253.11
#Sta/Elev= 30
  4345.7 1007.49  4389.3 1005.70  4407.0 1004.53  4465.7 1002.83  4476.6 1002.94
  4558.5 1001.20  4640.2 1000.59  4710.1  999.53  4809.2  996.99  4861.6  996.29
  4885.0  994.80  4891.0  995.09  4901.9  996.71  4922.3  996.81  4931.9  997.33
  4955.3  996.01  4967.4  994.64  4995.3  993.52  4995.6  990.52  4999.1  990.52
  4999.3  993.52  5002.5  993.52  5010.1  994.94  5020.1  995.27  5030.1  996.69
  5041.5  997.52  5079.0 1001.17  5084.0 1000.95  5090.3 1002.16  5150.5 1004.04
#Mann=5,-1,0
  4345.7    0.05       0  4922.3    0.12       0  4995.3    0.07       0
  4999.3    0.12       0  5041.5    0.05       0
Bank Sta=4995.3,4999.3
Exp/Cntr=0.3,0.1

Type RM Length L Ch R = 1,18739,475,475,475
BEGIN DESCRIPTION:
SANDY CREEK 35.0
END DESCRIPTION:
XS GIS Cut Line= 3
      2878305.69     10243353.12      2877482.25     10242854.00
      2876755.71     10243153.10
#Sta/Elev= 30
  4037.1 1014.61  4283.4 1005.36  4626.6 1000.43  4642.1  999.52  4669.3 1000.05
  4737.1  998.97  4822.4  999.01  4917.4  997.21  4931.4  994.61  4948.4  991.64
  4954.3  992.01  4958.8  991.10  4959.1  988.10  4962.8  988.10  4963.1  991.10
  4969.8  991.94  5006.2  991.50  5059.6  995.23  5072.0  994.67  5112.9  996.22
  5126.1  995.16  5171.6  995.87  5201.8  995.21  5356.7  998.85  5427.3 1001.53
  5547.8 1004.19  5601.9 1006.93  5688.4 1009.16  5723.2 1010.91  5785.7 1012.12
#Mann=5,-1,0
  4037.1    0.05       0  4931.4    0.12       0  4958.8    0.07       0
  4963.1    0.12       0  5356.7    0.05       0
Bank Sta=4958.8,4963.1
Exp/Cntr=0.3,0.1

Type RM Length L Ch R = 1,18264,494,494,494
BEGIN DESCRIPTION:
SANDY CREEK 34.0
END DESCRIPTION:
XS GIS Cut Line= 3
      2877852.71     10242611.71      2877441.75     10242382.00
      2876805.72     10242653.10
#Sta/Elev= 30
  4529.2  999.55  4571.1  999.16  4804.7  996.03  4812.2  995.17  4820.7  995.73
  4864.7  994.30  4885.8  993.77  4929.2  989.54  4961.1  990.48  4966.9  989.58
  4972.6  989.75  4986.4  987.22  4986.7  984.22  4990.5  984.22  4990.8  987.22
  5006.6  988.97  5013.8  991.68  5027.8  992.48  5202.3  994.94  5213.1  994.43
  5319.0  994.94  5348.1  996.84  5365.3  996.11  5412.8  996.93  5430.5  997.79
  5448.0  997.33  5484.9  998.20  5577.0 1001.47  5624.2 1004.17  5691.4 1006.11
#Mann=7,-1,0
  4529.2    0.05       0  4571.1    0.12       0  4864.7    0.05       0
  4986.4    0.05       0  4990.8    0.05       0  5027.8    0.12       0
  5412.8    0.05       0
Bank Sta=4986.4,4990.8
Exp/Cntr=0.3,0.1

Type RM Length L Ch R = 1,17770,473,473,473
BEGIN DESCRIPTION:
SANDY CREEK 33.0
END DESCRIPTION:
XS GIS Cut Line= 3
      2877842.96     10242061.71      2877216.75     10241950.00
      2876755.70     10242453.09
#Sta/Elev= 30
  4363.9  991.95  4380.4  992.48  4385.5  991.73  4422.1  994.26  4503.4  997.33
  4655.7  997.47  4724.1  996.13  4831.7  992.79  4858.9  991.50  4930.0  990.26
  4949.5  987.92  4954.6  988.53  4970.6  985.31  4990.9  985.53  4995.8  984.51
  4996.1  981.51  4999.9  981.51  5000.2  984.51  5004.5  984.51  5010.0  987.66
  5038.4  989.33  5073.5  988.92  5137.6  989.71  5229.5  992.94  5441.6  996.71
  5455.8  996.42  5505.8  998.86  5526.7  998.75  5610.3 1001.00  5682.4 1003.27
#Mann=6,-1,0
  4363.9    0.05       0  4724.1    0.12       0  4831.7    0.05       0
  4995.8    0.03       0  5000.2    0.05       0  5610.3    0.12       0
Bank Sta=4995.8,5000.2
Exp/Cntr=0.3,0.1

Type RM Length L Ch R = 1,17297,476,476,476
BEGIN DESCRIPTION:
SANDY CREEK 32.0
END DESCRIPTION:
XS GIS Cut Line= 3
      2877534.82     10241680.24      2877076.00     10241504.00
      2876755.69     10242053.10
#Sta/Elev= 30
  4508.5  990.75  4614.7  989.69  4623.0  990.16  4628.4  989.44  4653.0  990.31
  4683.0  990.22  4754.0  988.29  4871.7  987.76  4907.1  988.31  4937.1  987.71
  4956.4  984.68  4991.8  984.17  4995.3  983.53  4995.6  980.53  4999.4  980.53
  4999.7  983.53  5013.4  984.60  5029.2  983.80  5050.7  986.17  5056.0  985.99
  5189.6  987.86  5218.9  989.30  5232.6  990.90  5239.1  990.58  5248.3  990.35
  5285.5  992.25  5430.2  995.98  5445.9  995.57  5488.9  997.38  5635.7  999.39
#Mann=5,-1,0
  4508.5    0.05       0  4995.3    0.05       0  4999.7    0.05       0
  5056.0    0.12       0  5239.1    0.05       0
Bank Sta=4995.3,4999.7
Exp/Cntr=0.3,0.1

Type RM Length L Ch R = 1,16821,490,490,490
BEGIN DESCRIPTION:
SANDY CREEK 31.0
END DESCRIPTION:
XS GIS Cut Line= 3
      2877905.64     10241303.10      2876891.25     10241116.00
      2876155.64     10240903.10
#Sta/Elev= 30
  3968.5 1003.68  3994.9  999.91  4053.0  998.35  4106.0  994.43  4168.1  994.77
  4222.7  986.56  4270.1  981.79  4332.3  981.91  4333.6  982.04  4354.9  980.62
  4365.0  976.89  4372.8  976.71  4373.1  973.71  4377.3  973.71  4377.7  976.71
  4434.1  981.89  4519.3  982.92  4558.2  984.50  4792.1  982.88  4914.1  984.72
  4944.6  983.00  4965.0  984.10  5005.8  980.53  5047.4  986.84  5208.5  983.99
  5269.2  985.17  5370.7  982.15  5472.3  983.42  5690.2  995.46  5765.8  998.14
#Mann=11,-1,0
  3968.5    0.05       0  4168.1    0.12       0  4332.3    0.05       0
  4333.6    0.12       0  4372.8    0.05       0  4377.7    0.12       0
  4519.3    0.05       0  5269.2    0.12       0  5370.7    0.05       0
  5472.3    0.12       0  5690.2    0.05       0
Bank Sta=4372.8,4377.7
Exp/Cntr=0.3,0.1

Type RM Length L Ch R = 1,16331,467,467,467
BEGIN DESCRIPTION:
SANDY CREEK 30.0
END DESCRIPTION:
XS GIS Cut Line= 3
      2877705.73     10241053.13      2877097.50     10240787.00
      2876205.65     10240803.11
#Sta/Elev= 30
  4336.1  996.29  4408.9  993.46  4428.2  991.90  4534.0  983.33  4554.5  980.08
  4600.8  978.12  4609.0  975.99  4630.9  974.77  4641.8  976.31  4676.5  975.91
  4707.3  979.21  4746.6  980.52  4921.3  980.89  4944.6  979.52  4958.3  975.64
  4980.2  975.95  4994.4  974.10  4994.8  971.10  4999.0  971.10  4999.3  974.10
  5059.2  978.31  5091.8  977.68  5161.8  981.74  5331.9  982.03  5471.9  977.31
  5561.9  983.56  5651.9  985.77  5741.9  991.58  5849.7  994.90  5892.0  996.91
#Mann=7,-1,0
  4336.1    0.12       0  4408.9    0.05       0  4428.2    0.12       0
  4534.0    0.05       0  4994.4    0.05       0  4999.3    0.05       0
  5849.7    0.12       0
Bank Sta=4994.4,4999.3
Exp/Cntr=0.3,0.1

Type RM Length L Ch R = 1,15864,499,499,499
BEGIN DESCRIPTION:
SANDY CREEK 29.0
END DESCRIPTION:
XS GIS Cut Line= 3
      2877555.71     10240253.10      2877109.50     10240385.00
      2876305.68     10240753.11
#Sta/Elev= 30
  4534.7  987.52  4722.4  979.28  4826.7  970.81  4899.7  971.21  4920.6  974.55
  4943.5  975.23  4971.6  970.72  4991.1  969.45  4991.4  966.45  4995.7  966.45
  4996.1  969.45  5060.1  970.30  5092.2  970.44  5100.6  973.55  5106.1  971.96
  5114.2  976.20  5129.1  977.38  5170.9  977.64  5485.2  979.10  5499.1  978.54
  5513.7  973.78  5521.1  973.93  5559.7  977.75  5588.3  975.38  5605.8  978.39
  5686.1  985.33  5754.8  987.02  5772.3  988.96  5800.8  988.49  5884.1  992.80
#Mann=5,-1,0
  4534.7    0.05       0  4991.1    0.05       0  4996.1    0.05       0
  5060.1    0.12       0  5170.9    0.05       0
Bank Sta=4991.1,4996.1
Exp/Cntr=0.3,0.1

Type RM Length L Ch R = 1,15365,477,477,477
BEGIN DESCRIPTION:
SANDY CREEK 28.0
END DESCRIPTION:
XS GIS Cut Line= 3
      2877505.70     10239903.11      2877260.50     10239932.00
      2876455.70     10240553.10
#Sta/Elev= 30
  4753.1  981.77  4904.2  975.50  4924.3  972.73  4987.5  968.14  5011.2  967.51
  5032.0  969.10  5078.0  965.16  5078.5  962.16  5085.3  962.16  5085.8  965.16
  5096.3  968.24  5110.8  970.26  5154.3  973.04  5258.5  974.68  5344.3  973.95
  5384.0  974.29  5453.2  975.86  5608.6  974.32  5623.8  973.84  5667.0  973.93
  5675.2  970.95  5681.5  972.01  5688.2  969.68  5830.9  977.11  5888.9  977.64
  5895.2  975.13  5909.7  972.75  5953.2  975.02  5974.1  978.77  6016.6  981.90
#Mann=9,-1,0
  4753.1    0.05       0  4987.5    0.12       0  5078.0    0.07       0
  5085.8    0.12       0  5258.5    0.05       0  5344.3    0.12       0
  5384.0    0.05       0  5608.6    0.12       0  5623.8    0.05       0
Bank Sta=5078,5085.8
Exp/Cntr=0.3,0.1

Type RM Length L Ch R = 1,14888,479,479,479
BEGIN DESCRIPTION:
SANDY CREEK 27.0
END DESCRIPTION:
XS GIS Cut Line= 3
      2877405.70     10239503.11      2877013.50     10239560.00
      2876205.67     10240353.13
#Sta/Elev= 30
  4603.7  985.69  4635.6  984.45  4684.5  978.92  4805.8  968.92  4846.8  968.15
  4876.5  966.71  4906.9  968.72  4962.1  967.10  4977.6  964.56  4991.6  964.96
  5006.1  964.70  5018.0  964.48  5018.5  961.48  5025.4  961.48  5025.9  964.48
  5057.2  966.36  5071.3  969.94  5135.1  971.31  5255.2  971.52  5311.8  969.53
  5342.5  966.47  5361.3  966.51  5375.4  968.20  5382.5  971.26  5396.7  972.46
  5460.2  973.38  5502.7  971.37  5573.4  973.64  5778.5  975.04  6132.1  988.91
#Mann=9,-1,0
  4603.7    0.05       0  4635.6    0.12       0  4846.8    0.05       0
  4962.1    0.12       0  4991.6    0.05       0  5006.1    0.12       0
  5018.0    0.05       0  5025.9    0.12       0  5342.5    0.05       0
Bank Sta=5018,5025.9
Exp/Cntr=0.3,0.1

Type RM Length L Ch R = 1,14409,470,470,470
BEGIN DESCRIPTION:
SANDY CREEK 26.0
END DESCRIPTION:
XS GIS Cut Line= 3
      2877405.71     10239403.13      2876994.75     10239104.00
      2876255.68     10239403.11
#Sta/Elev= 30
  4491.7  982.98  4606.3  977.94  4619.9  976.90  4742.3  968.53  4763.7  967.65
  4892.4  967.49  4907.1  965.52  4963.5  963.87  4982.0  960.53  4982.5  957.53
  4990.5  957.53  4991.0  960.53  5007.7  961.84  5085.3  962.73  5096.2  964.99
  5120.3  965.89  5139.0  964.06  5144.4  965.00  5160.8  962.39  5192.7  961.81
  5214.8  964.57  5267.1  966.27  5311.8  967.65  5391.5  966.73  5568.0  968.10
  5613.9  965.76  5704.8  970.00  5728.9  973.64  5782.5  976.37  5797.3  978.30
#Mann=9,-1,0
  4491.7    0.05       0  4606.3    0.12       0  4619.9    0.05       0
  4742.3    0.12       0  4763.7    0.05       0  4982.0    0.05       0
  4991.0    0.05       0  5267.1    0.12       0  5391.5    0.05       0
Bank Sta=4982,4991
Exp/Cntr=0.3,0.1

Type RM Length L Ch R = 1,13939,498,498,498
BEGIN DESCRIPTION:
SANDY CREEK 25.0
END DESCRIPTION:
XS GIS Cut Line= 3
      2877255.69     10238553.11      2876800.25     10238725.00
      2876205.69     10239103.11
#Sta/Elev= 30
  4513.2  973.21  4532.5  972.59  4608.2  969.28  4644.8  965.61  4673.9  964.10
  4684.2  962.13  4698.8  966.09  4748.4  966.90  4814.2  964.14  4833.7  964.58
  4863.9  959.87  4876.6  959.38  4908.7  960.17  4984.7  959.64  5002.9  958.47
  5008.6  959.90  5017.3  960.07  5029.7  958.68  5066.1  959.54  5075.5  958.84
  5076.8  957.90  5077.3  954.90  5085.4  954.90  5085.9  957.90  5175.4  963.07
  5457.4  964.02  5560.7  967.80  5609.8  970.73  5697.0  972.70  5704.6  973.97
#Mann=5,-1,0
  4513.2    0.05       0  4532.5    0.12       0  4644.8    0.05       0
  5076.8    0.03       0  5085.9    0.05       0
Bank Sta=5076.8,5085.9
Exp/Cntr=0.3,0.1

Type RM Length L Ch R = 1,13441,491,491,491
BEGIN DESCRIPTION:
SANDY CREEK 24.0
END DESCRIPTION:
XS GIS Cut Line= 3
      2877155.64     10238303.12      2876454.00     10238400.00
      2876055.71     10238303.12
#Sta/Elev= 30
  4291.7  972.62  4404.5  968.63  4453.2  966.17  4483.5  963.10  4513.7  961.53
  4523.8  961.34  4548.3  963.41  4625.2  962.83  4634.9  961.79  4645.0  962.86
  4675.3  962.89  4826.7  961.42  4840.9  961.11  4872.5  955.80  4873.0  952.80
  4881.4  952.80  4881.9  955.80  4887.3  957.66  4897.4  958.73  4927.6  960.18
  4968.0  958.51  4989.7  956.28  5010.8  955.85  5029.1  956.72  5060.0  960.01
  5101.2  959.27  5172.7  960.33  5255.6  964.28  5308.2  968.24  5409.9  971.88
#Mann=3,-1,0
  4291.7    0.05       0  4872.5    0.03       0  4881.9    0.05       0
Bank Sta=4872.5,4881.9
Exp/Cntr=0.3,0.1

Type RM Length L Ch R = 1,12950,499,499,499
BEGIN DESCRIPTION:
SANDY CREEK 23.0
END DESCRIPTION:
XS GIS Cut Line= 3
      2877155.73     10238253.13      2876428.25     10237937.00
      2876105.68     10237753.11
#Sta/Elev= 30
  4206.8  972.38  4359.5  966.99  4403.1  965.23  4419.8  963.82  4512.1  961.56
  4746.4  959.04  4769.9  957.62  4822.2  957.53  4869.1  958.50  4892.6  957.85
  4973.8  958.02  4981.0  956.63  4995.2  951.04  4995.7  948.04  5004.2  948.04
  5004.7  951.04  5019.1  951.59  5034.9  953.68  5040.7  953.01  5062.3  953.54
  5078.1  955.73  5083.9  954.98  5094.0  955.76  5115.6  955.12  5129.6  953.61
  5174.7  953.12  5180.4  953.91  5196.3  960.83  5210.1  962.17  5371.3  969.48
#Mann=3,-1,0
  4206.8    0.05       0  4995.2    0.05       0  5004.7    0.05       0
Bank Sta=4995.2,5004.7
Exp/Cntr=0.3,0.1

Type RM Length L Ch R = 1,12451,471,471,471
BEGIN DESCRIPTION:
SANDY CREEK 22.0
END DESCRIPTION:
XS GIS Cut Line= 3
      2877155.67     10237753.11      2876364.00     10237462.00
      2876155.69     10237453.11
#Sta/Elev= 30
  4156.5  969.63  4252.4  966.82  4318.7  963.50  4343.9  961.48  4444.2  956.96
  4521.4  955.73  4785.1  955.70  4804.8  954.66  4810.1  955.19  4835.2  952.69
  4840.6  953.45  4859.7  952.07  4881.0  952.86  4913.0  950.15  4944.9  950.53
  4957.1  949.52  4976.9  950.62  5000.0  949.23  5003.5  948.34  5004.0  945.34
  5012.6  945.34  5013.1  948.34  5028.3  948.61  5038.4  951.54  5058.4  951.54
  5078.4  952.60  5087.3  955.43  5092.3  954.38  5128.4  958.99  5208.5  964.27
#Mann=3,-1,0
  4156.5    0.05       0  5003.5    0.05       0  5013.1    0.05       0
Bank Sta=5003.5,5013.1
Exp/Cntr=0.3,0.1

Type RM Length L Ch R = 1,11980,476,476,476
BEGIN DESCRIPTION:
SANDY CREEK 21.0
END DESCRIPTION:
XS GIS Cut Line= 3
      2877255.69     10237703.11      2876451.50     10237002.00
      2876105.70     10237003.11
#Sta/Elev= 30
  3933.1  971.24  4188.0  962.96  4372.2  954.23  4549.7  952.18  4620.9  952.98
  4727.2  951.24  4847.8  951.65  4861.8  951.16  4875.3  948.78  4882.9  946.28
  4903.8  945.07  4925.7  948.70  4960.8  948.83  4981.6  946.77  4984.2  943.70
  4984.7  940.70  4993.8  940.70  4994.3  943.70  4995.3  944.71  5005.8  944.41
  5035.8  948.73  5055.8  949.44  5075.8  946.64  5085.8  946.83  5095.8  948.92
  5145.8  946.21  5165.8  950.73  5195.8  954.21  5285.8  958.43  5345.8  960.09
#Mann=3,-1,0
  3933.1    0.05       0  4984.2    0.03       0  4994.3    0.05       0
Bank Sta=4984.2,4994.3
Exp/Cntr=0.3,0.1

Type RM Length L Ch R = 1,11504,475,475,475
BEGIN DESCRIPTION:
SANDY CREEK 20.0
END DESCRIPTION:
XS GIS Cut Line= 3
      2877005.65     10236903.08      2876685.75     10236602.00
      2876105.65     10236603.11
#Sta/Elev= 30
  4560.7  953.78  4624.4  950.35  4681.0  948.92  4893.0  946.20  4907.2  945.10
  4914.5  943.03  4935.5  943.37  4942.8  945.20  4963.8  946.22  4971.1  945.64
  4985.3  942.51  5030.1  942.94  5035.0  941.34  5035.5  938.34  5044.6  938.34
  5045.1  941.34  5060.1  941.59  5090.1  945.50  5130.1  946.06  5160.1  944.69
  5180.1  942.50  5230.1  945.89  5270.1  943.38  5280.1  944.17  5310.1  949.45
  5320.1  950.05  5420.1  953.85  5460.1  954.56  5570.1  959.85  5580.1  959.69
#Mann=3,-1,0
  4560.7    0.05       0  5035.0    0.03       0  5045.1    0.05       0
Bank Sta=5035,5045.1
Exp/Cntr=0.3,0.1

Type RM Length L Ch R = 1,11029,470,470,470
BEGIN DESCRIPTION:
SANDY CREEK 19.0
END DESCRIPTION:
XS GIS Cut Line= 3
      2877055.71     10236253.12      2876692.00     10236152.00
      2876005.70     10236203.11
#Sta/Elev= 30
  4622.5  953.45  4713.3  949.40  4718.5  949.86  4752.7  947.70  4792.2  946.80
  4799.0  945.85  4850.9  944.51  4913.1  944.24  4954.7  942.03  4965.0  940.81
  4973.7  938.77  4980.6  938.08  4981.1  935.08  4990.5  935.08  4991.0  938.08
  5026.4  939.34  5036.4  941.49  5046.4  942.08  5066.5  941.86  5086.9  938.83
  5116.6  942.59  5126.7  942.88  5146.7  942.20  5166.8  942.76  5186.8  944.93
  5277.1  949.37  5377.4  951.76  5537.8  958.98  5557.9  960.29  5688.2  965.51
#Mann=3,-1,0
  4622.5    0.05       0  4980.6    0.03       0  4991.0    0.05       0
Bank Sta=4980.6,4991
Exp/Cntr=0.3,0.1

Type RM Length L Ch R = 1,10559,415,415,415
BEGIN DESCRIPTION:
SANDY CREEK 18.0
END DESCRIPTION:
XS GIS Cut Line= 3
      2877105.67     10235753.11      2876714.00     10235683.00
      2876005.69     10235703.11
#Sta/Elev= 30
  4602.1  957.41  4612.2  957.63  4629.0  955.73  4825.6  943.40  4859.3  942.84
  4866.2  941.95  4906.9  940.44  4927.2  936.30  4937.3  935.83  4971.9  937.42
  4982.9  934.96  4983.4  931.96  4992.9  931.96  4993.4  934.96  4996.6  936.49
  5000.0  936.49  5008.3  939.01  5018.3  939.76  5098.4  940.80  5128.4  939.25
  5138.4  936.55  5148.4  937.24  5158.4  939.50  5176.7  941.60  5188.4  942.02
  5218.4  942.69  5308.4  942.51  5428.5  945.64  5498.5  948.95  5708.6  961.80
#Mann=3,-1,0
  4602.1    0.05       0  4982.9    0.05       0  4993.4    0.05       0
Bank Sta=4982.9,4993.4
Exp/Cntr=0.3,0.1

Type RM Length L Ch R = 1,10144,326,326,326
BEGIN DESCRIPTION:
Mapping XS ae5aaec2
END DESCRIPTION:
XS GIS Cut Line= 3
      2877784.75     10235291.33      2876555.61     10235291.33
      2875660.25     10235291.33
#Sta/Elev= 30
  4043.3  948.79  4082.4  952.08  4192.4  951.95  4512.4  941.47  4602.4  942.40
  4682.4  939.39  4722.4  936.28  4762.4  942.13  4932.4  941.40  4942.4  940.93
  4962.4  934.42  4972.4  933.66  5012.4  934.64  5032.4  938.20  5052.4  936.47
  5102.4  939.50  5192.4  936.54  5217.1  933.24  5217.6  930.24  5227.1  930.24
  5227.6  933.24  5252.4  939.76  5382.4  938.83  5582.4  940.07  5692.4  944.12
  5832.4  953.20  5902.4  955.68  5992.4  951.46  6132.4  941.11  6167.8  943.99
#Mann=3,-1,0
  4043.3    0.05       0  5217.1    0.03       0  5227.6    0.05       0
Bank Sta=5217.1,5227.6
Exp/Cntr=0.3,0.1

Type RM Length L Ch R = 1,9818,433,433,433
BEGIN DESCRIPTION:
Mapping XS 619bc3f0
END DESCRIPTION:
XS GIS Cut Line= 4
      2877638.94     10234999.67      2876597.27     10234978.83
      2875680.61     10235020.50      2875348.84     10235269.33
#Sta/Elev= 30
  4119.2  958.41  4182.5  957.03  4422.5  942.58  4482.5  944.09  4582.5  939.17
  4682.6  938.29  4692.3  939.50  4702.6  943.62  4752.6  945.68  4922.6  938.24
  4996.7  930.84  4997.2  927.84  5008.0  927.84  5008.5  930.84  5032.6  935.71
  5052.6  937.08  5102.6  935.53  5122.7  931.93  5192.7  938.15  5443.0  936.20
  5581.9  937.17  5683.2  939.81  5802.1  946.40  5807.1  945.05  5913.4  946.76
  6027.3  942.81  6155.8  944.50  6212.1  940.82  6291.2  945.29  6493.4  948.20
#Mann=3,-1,0
  4119.2    0.05       0  4996.7    0.05       0  5008.5    0.05       0
Bank Sta=4996.7,5008.5
Exp/Cntr=0.3,0.1

Type RM Length L Ch R = 1,9385,741,741,741
BEGIN DESCRIPTION:
Mapping XS b08d1f7f
END DESCRIPTION:
XS GIS Cut Line= 3
      2876909.79     10234332.98      2876513.94     10234666.33
      2875849.02     10234832.56
#Sta/Elev= 30
  4622.2  942.07  4632.1  943.54  4703.6  940.96  4759.6  944.20  4816.8  944.08
  4866.2  939.01  4880.5  935.47  4888.3  931.63  4894.8  931.00  4896.2  929.49
  4896.7  926.49  4907.6  926.49  4908.1  929.49  4944.3  933.12  4952.0  932.12
  4958.6  933.31  4966.3  930.24  4993.7  929.75  5008.0  929.64  5022.3  931.66
  5058.7  931.09  5065.2  932.26  5100.3  931.02  5108.1  933.66  5122.4  935.33
  5158.5  936.39  5498.7  934.35  5570.8  935.14  5777.0  944.91  5825.1  945.99
#Mann=3,-1,0
  4622.2    0.05       0  4896.2    0.05       0  4908.1    0.05       0
Bank Sta=4896.2,4908.1
Exp/Cntr=0.3,0.1

Type RM Length L Ch R = 1,8644,460,460,460
BEGIN DESCRIPTION:
SANDY CREEK 14.0
END DESCRIPTION:
XS GIS Cut Line= 3
      2876355.67     10233653.15      2876215.50     10233965.00
      2875705.70     10234753.08
#Sta/Elev= 30
  4658.1  946.41  4690.1  944.29  4718.7  941.04  4800.6  935.50  4822.5  934.87
  4840.0  932.97  4868.6  931.72  4886.3  932.33  4932.1  931.68  4938.1  932.68
  4954.1  931.73  4976.0  927.53  4996.2  925.12  5033.5  926.40  5069.6  925.88
  5072.8  924.65  5073.3  921.65  5084.3  921.65  5084.8  924.65  5105.9  926.77
  5128.8  931.71  5136.2  932.42  5172.5  932.85  5229.9  931.71  5245.1  932.50
  5359.8  930.34  5504.9  931.82  5605.2  935.67  5650.0  936.45  5938.6  947.85
#Mann=3,-1,0
  4658.1    0.05       0  5072.8    0.05       0  5084.8    0.05       0
Bank Sta=5072.8,5084.8
Exp/Cntr=0.3,0.1

Type RM Length L Ch R = 1,8184,478,478,478
BEGIN DESCRIPTION:
SANDY CREEK 13.0
END DESCRIPTION:
XS GIS Cut Line= 3
      2875855.69     10233653.09      2875804.50     10233782.00
      2875655.70     10234153.08
#Sta/Elev= 30
  4861.3  938.34  4876.2  937.57  4900.5  932.69  4905.8  932.57  4924.8  928.57
  4930.2  928.20  4936.6  924.84  4948.8  922.75  4954.5  921.78  4968.9  921.57
  4972.7  920.87  4973.2  917.87  4984.4  917.87  4984.9  920.87  4990.4  921.82
  5008.4  921.05  5044.3  922.84  5055.1  924.16  5062.2  925.88  5076.6  927.84
  5086.4  928.45  5152.0  928.31  5162.8  929.31  5169.8  931.17  5175.2  932.06
  5205.9  933.51  5238.2  932.71  5282.8  935.24  5385.0  937.04  5399.8  936.95
#Mann=4,-1,0
  4861.3    0.12       0  4948.8    0.05       0  4972.7    0.05       0
  4984.9    0.05       0
Bank Sta=4972.7,4984.9
Exp/Cntr=0.3,0.1

Type RM Length L Ch R = 1,7706,410,410,410
BEGIN DESCRIPTION:
SANDY CREEK 12.0
END DESCRIPTION:
XS GIS Cut Line= 3
      2875605.70     10233453.10      2875370.25     10233667.00
      2875505.66     10233953.07
#Sta/Elev= 30
  4681.9  943.18  4745.8  938.09  4766.7  934.73  4774.2  934.40  4788.3  931.29
  4809.3  928.63  4816.7  928.53  4823.5  926.82  4845.4  926.35  4866.1  925.56
  4880.2  921.55  4887.0  918.13  4922.8  918.53  4923.5  916.76  4924.0  913.76
  4935.2  913.76  4935.7  916.76  4937.0  917.72  4943.8  918.70  4958.0  917.44
  5006.8  917.35  5040.0  918.63  5084.2  922.38  5092.1  924.35  5097.7  923.94
  5114.9  927.99  5128.5  928.75  5239.7  932.15  5256.9  931.59  5316.5  933.00
#Mann=4,-1,0
  4681.9    0.12       0  4845.4    0.05       0  4923.5    0.03       0
  4935.7    0.05       0
Bank Sta=4923.5,4935.7
Exp/Cntr=0.3,0.1

Type RM Length L Ch R = 1,7296,499,499,499
BEGIN DESCRIPTION:
SANDY CREEK 11.0
END DESCRIPTION:
XS GIS Cut Line= 3
      2875305.68     10233203.12      2874996.25     10233605.00
      2874605.68     10233703.11
#Sta/Elev= 30
  4492.8  932.46  4620.5  925.76  4693.0  924.09  4707.3  925.27  4720.2  923.49
  4737.6  923.00  4778.0  925.14  4828.0  924.94  4871.4  923.11  4901.0  924.45
  4927.7  923.43  4934.5  922.29  4948.5  916.93  4985.0  915.37  4989.4  914.37
  4989.9  911.37  5002.9  911.37  5003.4  914.37  5050.4  920.56  5055.6  922.74
  5062.4  923.80  5103.7  925.06  5132.7  923.47  5137.8  924.20  5155.2  923.75
  5173.8  925.69  5179.0  924.56  5248.0  927.20  5343.6  928.52  5402.7  930.84
#Mann=6,-1,0
  4492.8    0.12       0  4737.6    0.05       0  4778.0    0.12       0
  4901.0    0.05       0  4989.4    0.05       0  5003.4    0.05       0
Bank Sta=4989.4,5003.4
Exp/Cntr=0.3,0.1
