--- MAGILL CREEK.prj (project) ---

Proj Title=MAGILL CREEK Base Level Engineering
Current Plan=p01
Default Exp/Contr=0.3,0.1
English Units
Geom File=g01
Flow File=f01
Plan File=p01
Y Axis Title=Elevation
X Axis Title(PF)=Main Channel Distance
X Axis Title(XS)=Station
BEGIN DESCRIPTION:
MAGILL CREEK
END DESCRIPTION:
DSS Export Rating Curves= 0
DSS Export Rating Curve Sorted= 0
DSS Export Volume Flow Curves= 0
DXF OffsetX= 0
DXF OffsetY= 0
DXF ScaleX= 1
DXF ScaleY= 10

--- MAGILL CREEK.p01 (plan) ---

Plan Title=Multiple Run
Short Identifier=Multiple
Geom File=g01
Flow File=f01
Subcritical Flow
K Sum by GR= 0
Std Step Tol= 0.01
Critical Tol= 0.01
Num of Std Step Trials= 20
Max Error Tol= 0.3
Flow Tol Ratio= 0.001
Split Flow NTrial= 30
Split Flow Tol= 0.02
Split Flow Ratio= 0.02
Log Output Level= 0
Friction Slope Method= 1
Unsteady Friction Slope Method= 2
Unsteady Bridges Friction Slope Method= 1
Parabolic Critical Depth
Global Vel Dist=  1 , 1 , 1
Global Log Level= 0
CheckData=True
Encroach Param= -1, 0, 0, 0
BEGIN DESCRIPTION:
Multiple Run
END DESCRIPTION:

--- MAGILL CREEK.f01 (steady flow) ---

Flow Title=Multiple
Number of Profiles=7
Profile Names=10-year,25-year,50-year,1pct_min,100-year,1pct_plu,500-year
River Rch & RM= MAGILL CREEK,Reach-1,24500
     417     672    1261     897    1749    3412    2511
River Rch & RM= MAGILL CREEK,Reach-1,15500
     763    1285    2417    1752    3420    6676    4901
River Rch & RM= MAGILL CREEK,Reach-1,8000
    1024    1760    3291    2047    4693   10757    6694
River Rch & RM= MAGILL CREEK,Reach-1,3500
    1200    2086    3839    2284    5493   13206    7813
Boundary for River Rch & Prof#=MAGILL CREEK,Reach-1,1
Up Type=0
Dn Type=3
Dn Slope=0.005
Boundary for River Rch & Prof#=MAGILL CREEK,Reach-1,2
Up Type=0
Dn Type=3
Dn Slope=0.005
Boundary for River Rch & Prof#=MAGILL CREEK,Reach-1,3
Up Type=0
Dn Type=3
Dn Slope=0.005
Boundary for River Rch & Prof#=MAGILL CREEK,Reach-1,4
Up Type=0
Dn Type=3
Dn Slope=0.005
Boundary for River Rch & Prof#=MAGILL CREEK,Reach-1,5
Up Type=0
Dn Type=3
Dn Slope=0.005
Boundary for River Rch & Prof#=MAGILL CREEK,Reach-1,6
Up Type=0
Dn Type=3
Dn Slope=0.005
Boundary for River Rch & Prof#=MAGILL CREEK,Reach-1,7
Up Type=0
Dn Type=3
Dn Slope=0.005

--- MAGILL CREEK.g01 (geometry) ---

Geom Title=Existing Conditions
Program Version=4.10

River Reach=MAGILL CREEK    ,Reach-1
Reach XY= 30
      2784312.75       10295750.        2783766.       10295497.
      2783226.75       10294786.      2783642.25       10293165.
      2785121.25       10292696.      2785385.75       10291847.
        2785585.       10291768.      2785609.75       10291312.
      2786381.75       10290563.        2786891.       10290392.
        2787189.       10289842.      2788056.25       10289558.
        2788384.       10288565.      2788915.25       10288603.
      2789101.75       10288035.       2788405.5       10287406.
      2788448.75       10286915.        2789730.       10286310.
       2790064.5       10285906.      2790148.75       10285249.
      2790575.75       10284909.      2791909.25       10284509.
      2792267.75       10284635.      2793131.25       10284415.
      2793256.25       10284828.      2793447.25       10284879.
       2795667.5       10284925.        2796822.       10285484.
      2797348.25       10285460.       2797583.5       10285252.

Type RM Length L Ch R = 1 ,24500   ,500,500,500
BEGIN DESCRIPTION:
MAGILL CREEK 49.0
END DESCRIPTION:
XS GIS Cut Line= 3
      2784155.66     10295353.13      2783923.52     10295553.57
      2783705.71     10295803.08
#Sta/Elev= 30
  4693.3 1567.74  4696.6 1567.74    4707 1562.25  4721.3  1557.5  4778.9 1540.57
  4821.1 1529.26  4835.3 1527.06  4849.6 1522.12  4948.3 1514.52  4962.6 1511.11
  4970.2 1511.21  4974.8 1507.74  4975.1 1507.24  4978.8 1507.74  4991.1  1509.7
  5005.2 1507.84  5012.7  1512.4    5026  1514.4    5083 1515.43  5097.2 1514.01
  5111.5  1515.4    5140 1526.67  5168.4  1535.4  5203.6 1542.99    5232 1552.43
  5267.2 1557.82  5295.6  1568.1  5317.5 1579.38  5327.9 1583.29  5331.2 1583.29
#Mann= 4 ,-1 , 0
  4693.3     .12       0  4778.9     .05       0  4974.8     .05       0
  4978.8     .05       0
Bank Sta=4974.8,4978.8
XS Rating Curve= 0 ,0
Exp/Cntr=0.3,0.1

Type RM Length L Ch R = 1 ,24000   ,500,500,500
BEGIN DESCRIPTION:
MAGILL CREEK 48.0
END DESCRIPTION:
XS GIS Cut Line= 3
      2783805.66     10295053.13      2783558.64     10295258.27
      2783355.71     10295653.07
#Sta/Elev= 30
  4678.9 1565.61  4682.1 1565.61  4706.9  1554.2  4735.5  1546.4  4778.5 1529.28
  4835.3 1512.22  4863.1 1505.55  4919.6 1500.28  4969.9 1498.55  4981.4 1494.96
  4988.8  1490.2  4989.1  1489.7  4992.8  1490.2  5036.4  1496.1    5042 1493.95
  5064.2 1493.43    5103 1498.77  5125.1 1500.18  5152.9 1498.99  5175.1 1500.32
  5219.5 1506.24    5236 1511.42  5280.4 1521.42  5286.5 1524.55  5302.6 1528.61
  5346.9 1545.06    5354 1549.97  5391.3 1560.44  5407.9 1569.07  5443.9 1579.78
#Mann= 6 ,-1 , 0
  4678.9     .12       0  4835.3     .05       0  4919.6     .12       0
  4981.4     .05       0  4988.8     .05       0  4992.8     .05       0
Bank Sta=4988.8,4992.8
XS Rating Curve= 0 ,0
Exp/Cntr=0.3,0.1

Type RM Length L Ch R = 1 ,23500   ,177,177,177
BEGIN DESCRIPTION:
MAGILL CREEK 47.0
END DESCRIPTION:
XS GIS Cut Line= 3
      2783655.69     10294953.11      2783267.18      10294871.4
      2782755.71      10295253.1
#Sta/Elev= 30
    4603 1531.11  4622.8 1523.04  4627.9 1524.17  4633.7 1520.43  4646.2 1517.14
    4695 1503.42    4750 1493.23  4804.6 1488.21  4981.1 1479.22  4991.3 1477.79
  4996.2 1474.16  4996.5 1473.66  5000.2 1474.16  5030.5 1476.32  5045.1  1478.6
  5051.8 1476.01  5065.9 1474.85  5074.3 1478.57  5088.9 1481.15  5162.6 1485.04
  5261.4 1492.09  5295.6 1494.45    5465 1507.37  5488.5 1511.28    5510 1517.93
  5530.9 1521.02  5580.9 1534.55    5630 1551.89  5635.1 1555.39  5638.2 1555.39
#Mann= 11 ,-1 , 0
    4603     .12       0  4646.2     .05       0    4750     .12       0
  4804.6     .05       0  4996.2     .05       0  5030.5     .05       0
  5162.6     .12       0  5261.4     .05       0  5295.6     .12       0
    5465     .05       0    5630     .12       0
#XS Ineff= 2 , 0
                         5045.77         1478.95
Permanent Ineff=
       F       F
Bank Sta=4996.2,5000.2
XS Rating Curve= 0 ,0
Exp/Cntr=0.3,0.1

Type RM Length L Ch R = 1 ,23323   ,323,323,323
BEGIN DESCRIPTION:
Mapping XS 19c45dc3
END DESCRIPTION:
XS GIS Cut Line= 3
      2783390.91     10294740.01       2783130.5     10294687.92
      2782740.31     10294791.97
#Sta/Elev= 30
  4819.4  1480.2  4866.4  1476.2  4916.5 1474.42  4957.3 1474.01  4967.5 1474.42
  4975.3 1473.55  4975.6 1473.05  4979.3 1473.55  4998.1 1473.86  5028.3 1473.78
  5038.9 1474.71  5049.1 1473.61  5066.2 1477.21  5079.3 1480.11  5084.4 1478.72
  5090.4 1479.58  5110.7 1478.09  5125.3 1478.65  5307.3 1494.14  5338.3 1498.68
  5360.8 1503.28  5375.8 1507.24  5390.1  1510.8  5395.7  1513.4  5400.9 1513.58
  5435.8 1521.41  5441.8 1523.97  5470.8 1532.94  5475.9 1533.79  5488.8 1540.61
#Mann= 6 ,-1 , 0
  4819.4     .05       0  4866.4     .12       0  4957.3     .05       0
  4998.1     .12       0  5066.2     .05       0  5375.8     .12       0
Bank Sta=4975.3,4979.3
XS Rating Curve= 0 ,0
Exp/Cntr=0.3,0.1

Type RM Length L Ch R = 1 ,23000   ,500,500,500
BEGIN DESCRIPTION:
MAGILL CREEK 46.0
END DESCRIPTION:
XS GIS Cut Line= 3
      2783655.68     10294853.11      2783270.53     10294455.45
      2782755.71     10294553.11
#Sta/Elev= 30
  4446.4 1533.43  4453.5 1532.67  4460.4 1528.86  4467.6 1528.83  4474.6 1524.87
  4495.9 1521.21  4545.3 1506.12  4566.6 1503.29  4583.3 1499.08  4616.1 1492.06
  4658.5 1486.04  4856.6 1472.79  4941.4 1467.64  4988.8 1459.84  4989.1 1459.34
  4992.8 1459.84    5005 1460.68  5012.2 1462.33  5017.2 1460.93  5035.5 1464.19
  5055.8 1462.96  5064.4 1463.86  5069.5 1462.03  5106.7 1468.76  5157.6 1471.29
  5401.9 1488.81  5473.1 1498.07  5492.8 1502.52  5503.7 1506.58    5524 1510.66
#Mann= 4 ,-1 , 0
  4446.4     .12       0  4583.3     .05       0  4856.6     .05       0
    5005     .05       0
#XS Ineff= 2 , 0
                         5041.38         1464.46
Permanent Ineff=
       F       F
Bank Sta=4988.8,4992.8
XS Rating Curve= 0 ,0
Exp/Cntr=0.3,0.1

Type RM Length L Ch R = 1 ,22500   ,185,185,185
BEGIN DESCRIPTION:
MAGILL CREEK 45.0
END DESCRIPTION:
XS GIS Cut Line= 3
      2783855.71     10294403.14      2783441.32      10293991.5
       2782605.7     10294353.11
#Sta/Elev= 30
  4415.9 1501.32  4419.6 1501.31  4458.3 1494.75  4465.4 1495.14  4472.5 1492.79
  4514.9 1486.94  4553.1 1483.94  4599.8 1477.74  4686.6 1470.84    4925 1456.71
  4953.3 1455.24  4988.7  1449.8  5004.1 1449.02  5004.4 1448.52  5008.1 1449.02
  5014.1 1451.82  5019.6    1450  5049.7 1455.26    5072  1455.4  5212.9 1457.15
  5241.8 1459.61  5485.6 1471.16  5545.5 1472.84  5597.9 1476.52  5749.7 1483.58
  5790.7 1481.83  5820.1 1487.79  5825.6 1486.77  5872.6  1494.3  5910.5 1496.94
#Mann= 7 ,-1 , 0
  4415.9     .05       0  4419.6     .12       0  4458.3     .05       0
  4553.1     .12       0  4686.6     .05       0    4925     .05       0
    5072     .05       0
Bank Sta=5004.1,5008.1
XS Rating Curve= 0 ,0
Exp/Cntr=0.3,0.1

Type RM Length L Ch R = 1 ,22315   ,588,588,588
BEGIN DESCRIPTION:
Mapping XS 5e9853bd
END DESCRIPTION:
XS GIS Cut Line= 3
       2783975.9      10294048.9      2783400.82     10293766.79
      2782783.52     10293918.41
#Sta/Elev= 30
  4509.4 1463.05  4535.7 1461.49  4642.6 1459.91  4654.4 1458.46  4665.1 1458.84
    4699 1456.64  4760.6 1455.25  4856.1 1451.34  4873.1 1451.73  4878.6 1450.54
    4918 1450.49    4963 1448.62  4991.1 1445.47  5030.5 1448.85  5103.5  1448.1
  5186.1 1450.64  5235.9 1449.05  5241.1 1449.71  5258.2 1446.62  5266.5 1443.42
  5266.8 1442.92  5270.5 1443.42  5277.5 1445.35  5282.6 1444.28  5299.4 1450.47
  5309.7 1451.17  5433.3 1454.96  5578.7 1461.96  5680.4  1464.3  5785.6 1470.38
#Mann= 3 ,-1 , 0
  4509.4     .05       0  5235.9     .05       0  5309.7     .05       0
#XS Ineff= 2 , 0
         5185.58 1450.68
Permanent Ineff=
       F       F
Bank Sta=5266.5,5270.5
XS Rating Curve= 0 ,0
Exp/Cntr=0.3,0.1

Type RM Length L Ch R = 1 ,21727   ,227,227,227
BEGIN DESCRIPTION:
Mapping XS d86a44e0
END DESCRIPTION:
XS GIS Cut Line= 4
      2783823.99     10293875.28      2783704.64     10293462.97
      2783509.33     10293289.36      2783228.91     10293159.94
#Sta/Elev= 30
  4406.8 1451.83  4527.7 1446.29  4606.9 1445.75  4690.1 1446.44  4706.1 1447.57
  4773.3 1446.82  4948.5 1437.35  4962.8 1436.08  4995.9    1429  4996.1  1428.5
  4999.9    1429  5019.6 1432.69  5040.5 1434.65  5054.7 1434.88  5062.1 1433.61
    5069 1429.88  5075.6 1429.62  5089.9 1430.64    5121  1435.3  5166.9 1436.64
  5172.4 1436.01  5195.4  1438.2  5218.3 1438.25  5223.8 1437.33  5269.7 1443.55
  5287.2 1444.12  5292.7 1445.91  5310.1  1446.9  5344.1 1451.47  5406.2 1457.24
#Mann= 3 ,-1 , 0
  4406.8     .05       0  4995.9     .05       0  4999.9     .05       0
#XS Ineff= 2 , 0
                         5054.55         1434.98
Permanent Ineff=
       F       F
Bank Sta=4995.9,4999.9
XS Rating Curve= 0 ,0
Exp/Cntr=0.3,0.1

Type RM Length L Ch R = 1 ,21500   ,500,500,500
BEGIN DESCRIPTION:
MAGILL CREEK 43.0
END DESCRIPTION:
XS GIS Cut Line= 3
      2783755.68     10293253.11      2783660.48     10293144.81
      2783305.66      10292953.1
#Sta/Elev= 30
  4855.8 1436.47  4859.1 1436.47  4862.9 1435.43  4869.6 1436.04  4891.4 1434.38
  4934.1 1430.14  4940.7 1430.62  4975.8 1428.39  4995.6 1424.91  4995.9 1424.41
  4999.4 1424.41  4999.6 1424.91  5012.6 1425.37  5040.2 1430.04  5050.7 1430.26
  5056.4 1431.69  5072.6 1431.44  5094.5 1433.76  5100.1 1433.18  5107.7 1434.42
  5130.5 1436.18  5175.9 1438.53  5203.9 1440.88    5210 1441.97  5247.7 1444.66
  5263.9 1447.12  5269.5 1447.09    5301  1451.8  5367.6 1457.56  5403.3 1459.44
#Mann= 3 ,-1 , 0
  4855.8     .05       0  4995.6     .05       0  4999.6     .05       0
Bank Sta=4995.6,4999.6
XS Rating Curve= 0 ,0
Exp/Cntr=0.3,0.1

Type RM Length L Ch R = 1 ,21000   ,500,500,500
BEGIN DESCRIPTION:
MAGILL CREEK 42.0
END DESCRIPTION:
XS GIS Cut Line= 3
      2783805.69     10293553.09      2784075.51      10292926.3
      2783555.69     10292553.12
#Sta/Elev= 30
  4317.6 1449.18  4408.1 1447.61  4513.5  1443.9  4589.8 1444.19  4796.6 1430.67
  4840.8 1425.39    4949 1422.84  4970.8 1420.49  4981.7  1420.5  4990.9 1417.19
  4991.2 1416.69  4994.9 1417.19    4999 1418.88    5010 1417.75  5016.1  1420.5
  5030.9  1419.1    5037 1423.06  5045.6 1423.47  5051.8 1426.33  5060.3 1426.17
  5066.5 1427.49  5095.9 1426.32  5152.4 1428.92  5167.2 1428.02  5253.1 1429.47
  5332.2 1431.92    5440 1437.04  5517.1 1441.19  5541.1 1441.27  5639.9  1445.9
#Mann= 5 ,-1 , 0
  4317.6     .05       0  4990.9     .05       0  4994.9     .05       0
    5440     .12       0  5541.1     .05       0
Bank Sta=4990.9,4994.9
XS Rating Curve= 0 ,0
Exp/Cntr=0.3,0.1

Type RM Length L Ch R = 1 ,20500   ,500,500,500
BEGIN DESCRIPTION:
MAGILL CREEK 41.0
END DESCRIPTION:
XS GIS Cut Line= 3
      2784405.69     10293403.07      2784472.22     10292982.81
      2784555.69     10292653.11
#Sta/Elev= 30
  4574.5 1432.37  4655.5 1427.35  4716.2 1425.42  4868.1    1418  4878.2 1418.33
    4925 1414.89  4959.2 1413.85  4985.3 1411.04  4985.6 1410.54  4989.3 1411.04
    5010 1413.04  5020.3 1412.23    5030 1412.93  5035.1 1415.12    5071 1414.24
  5092.5 1414.88  5102.8 1416.14  5133.8 1415.55  5144.1 1416.25  5158.1 1414.83
  5185.4 1416.84  5199.2 1415.91  5226.6 1416.75    5235 1417.95  5240.2 1417.46
  5267.9 1420.57  5281.2 1418.42  5292.3 1419.29  5322.2 1417.27  5340.1 1417.99
#Mann= 4 ,-1 , 0
  4574.5     .05       0  4985.3     .05       0  4989.3     .05       0
  5292.3     .12       0
Bank Sta=4985.3,4989.3
XS Rating Curve= 0 ,0
Exp/Cntr=0.3,0.1

Type RM Length L Ch R = 1 ,20000   ,500,500,500
BEGIN DESCRIPTION:
MAGILL CREEK 40.0
END DESCRIPTION:
XS GIS Cut Line= 3
      2784755.68     10293703.11      2784861.85     10292760.47
      2784355.68     10292553.11
#Sta/Elev= 30
  4051.4 1443.41  4061.5  1440.7  4091.3 1438.14  4096.4 1439.46  4202.3 1435.74
  4242.6 1428.16  4276.3 1428.39  4292.9  1432.2    4303 1432.23    4313 1427.95
  4333.2 1424.59  4361.2 1424.49  4366.3 1427.47  4383.5 1425.43  4413.7 1427.44
  4451.2 1424.58  4546.2 1423.53  4923.5 1410.19  4983.9    1405  4984.2  1404.5
  4987.9    1405  4990.9 1407.35  5003.7 1405.32  5012.1 1406.35  5049.9 1406.87
  5169.3 1414.79  5228.2 1415.66  5363.3  1418.6  5430.3 1422.99    5547 1426.17
#Mann= 7 ,-1 , 0
  4051.4     .05       0  4923.5     .12       0  4983.9     .07       0
  4987.9     .12       0  5012.1     .05       0  5228.2     .12       0
  5430.3     .05       0
Bank Sta=4983.9,4987.9
XS Rating Curve= 0 ,0
Exp/Cntr=0.3,0.1

Type RM Length L Ch R = 1 ,19500   ,500,500,500
BEGIN DESCRIPTION:
MAGILL CREEK 39.0
END DESCRIPTION:
XS GIS Cut Line= 3
      2785405.69     10293503.15      2785193.01     10292534.73
      2784205.71     10292303.12
#Sta/Elev= 30
  4008.5 1430.67  4069.6 1428.17  4081.9 1426.61  4120.6 1426.47  4125.7 1425.17
  4141.6 1425.73    4249 1422.29    4343 1419.62  4540.1 1413.15  4558.6 1412.65
  4594.3 1411.01  4622.8 1411.54  4858.3 1405.54  4950.5 1402.28  4996.3 1398.88
  4996.5 1398.38  5000.3 1398.88    5026 1403.04  5168.8  1404.8  5320.3 1408.84
  5418.1 1413.14  5438.9 1412.89  5465.7 1415.29  5531.4 1416.75  5598.2 1420.34
    5688 1422.52  5761.9 1424.52  5886.4 1428.61  5978.8 1433.44  6014.1 1435.43
#Mann= 14 ,-1 , 0
  4008.5     .12       0  4069.6     .05       0    4249     .12       0
    4343     .05       0  4540.1     .12       0  4558.6     .05       0
  4996.3     .05       0  5000.3     .05       0  5168.8     .12       0
  5320.3     .05       0    5688     .12       0  5761.9     .05       0
  5886.4     .12       0  5978.8     .05       0
Bank Sta=4996.3,5000.3
XS Rating Curve= 0 ,0
Exp/Cntr=0.3,0.1

Type RM Length L Ch R = 1 ,19000   ,500,500,500
BEGIN DESCRIPTION:
MAGILL CREEK 38.0
END DESCRIPTION:
XS GIS Cut Line= 3
      2786005.65     10292553.08      2785351.02     10292060.91
      2784855.67      10291553.1
#Sta/Elev= 30
    4181 1412.94    4270  1409.8  4417.3 1404.12  4616.7    1401  4657.2 1400.57
  4790.1 1399.17  4952.6 1397.58    4992 1392.59  4992.3 1392.09    4996 1392.59
  5044.6 1396.31  5080.1 1396.08  5094.2 1394.35  5101.2 1395.74  5143.7 1394.89
  5228.5 1401.36  5306.2 1405.47  5443.3 1408.87  5461.8 1408.79    5469 1410.44
  5483.1 1409.83  5497.3 1412.28  5504.3  1410.4  5511.4 1411.58  5539.7 1409.59
    5604 1411.14    5667 1412.53    5674 1415.94  5681.2 1413.74  5709.4 1413.34
#Mann= 9 ,-1 , 0
    4181     .05       0    4270     .12       0  4616.7     .05       0
  4657.2     .12       0  4790.1     .05       0    4992     .05       0
    4996     .05       0  5443.3     .12       0    5604     .05       0
Bank Sta=4992,4996
XS Rating Curve= 0 ,0
Exp/Cntr=0.3,0.1

Type RM Length L Ch R = 1 ,18500   ,500,500,500
BEGIN DESCRIPTION:
MAGILL CREEK 37.0
END DESCRIPTION:
XS GIS Cut Line= 3
      2786105.67      10292203.1      2785591.69     10291715.31
      2785105.66     10291653.11
#Sta/Elev= 30
  4291.4 1408.71  4482.5 1403.74    4546 1403.58  4574.3 1402.53  4666.2 1403.99
  4701.7  1405.6  4715.9 1405.27  4779.4 1408.41  4829.1 1407.26  4842.9 1405.86
  4850.2  1404.1  4871.2    1404  4927.9 1399.37  4949.3 1393.22  4970.3 1391.21
  4977.6 1389.54  5004.1 1387.87  5004.3 1387.37  5008.1 1387.87  5026.2 1390.21
  5059.1 1390.85  5086.7 1392.71    5127 1393.34  5167.4 1395.22  5218.5 1395.22
  5237.9 1397.72  5293.2 1400.31  5328.7  1403.8  5488.4 1409.86    5490 1409.86
#Mann= 4 ,-1 , 0
  4291.4     .05       0  5004.1     .05       0  5008.1     .05       0
  5488.4     .12       0
Bank Sta=5004.1,5008.1
XS Rating Curve= 0 ,0
Exp/Cntr=0.3,0.1

Type RM Length L Ch R = 1 ,18000   ,500,500,500
BEGIN DESCRIPTION:
MAGILL CREEK 36.0
END DESCRIPTION:
XS GIS Cut Line= 3
      2785905.66     10291503.09      2785658.36     10291261.68
      2785455.65      10291203.1
#Sta/Elev= 30
  4654.4 1402.82  4703.9 1401.36  4746.3 1399.09  4788.7 1396.23  4809.9 1395.35
  4852.3 1391.75  4887.8 1390.08  4894.8 1389.24  4937.2 1386.92  4944.3 1387.04
  4979.6 1384.74  4986.8 1384.71  4998.4 1382.53  5008.4 1382.17  5008.7 1381.67
  5012.2 1381.67  5012.4 1382.17  5015.6 1385.01    5034  1388.9    5044 1390.36
  5054.8 1393.55  5075.6 1396.48  5082.9 1398.02  5088.1 1398.23  5127.7 1403.36
  5155.3 1405.41  5160.5 1406.35  5179.7 1408.23  5188.9  1409.8    5211 1411.13
#Mann= 3 ,-1 , 0
  4654.4     .05       0  5008.4     .05       0  5012.4     .05       0
Bank Sta=5008.4,5012.4
XS Rating Curve= 0 ,0
Exp/Cntr=0.3,0.1

Type RM Length L Ch R = 1 ,17500   ,500,500,500
BEGIN DESCRIPTION:
MAGILL CREEK 35.0
END DESCRIPTION:
XS GIS Cut Line= 3
      2786105.68     10291303.07      2786019.52      10290922.3
      2785805.69     10290703.12
#Sta/Elev= 30
  4609.6 1400.08  4640.3 1401.73  4691.6 1401.76  4753.1 1400.72  4775.5    1399
  4886.4 1389.19  4902.9 1386.59    4908 1386.71  4946.1 1382.03  4951.2 1380.65
  4990.3  1376.6  4992.4 1376.39  4992.6 1375.89  4996.4 1376.39  5009.2 1378.78
  5054.5  1383.3  5065.8 1384.19  5072.8  1383.4    5080 1384.21    5087  1383.7
  5094.1 1384.92  5101.1 1384.41  5107.6 1385.71  5122.4 1387.14  5129.4 1386.53
  5150.7 1388.77    5186 1390.07  5228.4 1394.07  5249.7 1397.82  5306.2 1400.54
#Mann= 7 ,-1 , 0
  4609.6     .05       0  4775.5     .12       0  4990.3     .05       0
  4992.4     .05       0  4996.4     .05       0  5054.5     .12       0
  5107.6     .05       0
Bank Sta=4992.4,4996.4
XS Rating Curve= 0 ,0
Exp/Cntr=0.3,0.1

Type RM Length L Ch R = 1 ,17000   ,500,500,500
BEGIN DESCRIPTION:
MAGILL CREEK 34.0
END DESCRIPTION:
XS GIS Cut Line= 3
      2786755.69     10291003.12      2786371.56      10290580.5
      2786305.69     10290403.14
#Sta/Elev= 30
  4428.9 1390.96  4484.8 1391.89  4553.7  1392.2  4584.7 1390.48  4591.4 1388.76
    4613 1387.98  4632.8 1385.43  4662.4 1380.42  4669.8 1380.46  4676.6 1379.08
  4761.1 1374.34  4796.8 1371.18    4834 1374.55  4853.6 1377.14  4867.8 1376.72
  4896.2 1373.42  4952.9  1372.8  4959.7 1371.08  4992.9 1367.94  4993.1 1367.44
  4996.9 1367.94    5000 1367.94  5002.5 1370.01  5018.6 1372.28  5039.9 1380.37
  5062.5 1384.94  5082.6 1385.74  5093.6 1387.72  5143.7 1391.21  5189.2 1392.39
#Mann= 9 ,-1 , 0
  4428.9     .05       0  4484.8     .12       0  4553.7     .05       0
  4632.8     .12       0  4761.1     .05       0    4834     .12       0
  4992.9     .07       0  4996.9     .12       0  5062.5     .05       0
Bank Sta=4992.9,4996.9
XS Rating Curve= 0 ,0
Exp/Cntr=0.3,0.1

Type RM Length L Ch R = 1 ,16500   ,500,500,500
BEGIN DESCRIPTION:
MAGILL CREEK 33.0
END DESCRIPTION:
XS GIS Cut Line= 3
       2787105.7     10290503.12      2786838.29     10290425.32
      2786505.69     10290203.11
#Sta/Elev= 30
  4721.5 1393.87  4731.9 1393.93  4738.3 1391.54  4752.8 1388.54  4763.2 1384.35
    4777 1381.35  4810.5 1378.82  4825.7 1376.13  4849.3 1373.83  4867.3 1373.35
  4888.2 1371.15    4955 1367.55  4988.6 1363.49  4996.8 1359.31    4997 1358.81
  5000.8 1359.31  5017.1 1360.32  5032.1 1363.05  5100.1 1366.77  5119.2  1368.8
    5147 1373.93  5176.3 1377.28  5191.3 1377.45  5197.3 1378.81  5227.3 1381.44
  5233.3  1382.9  5242.3 1382.73  5263.3 1385.95  5316.8  1391.9    5400 1400.36
#Mann= 6 ,-1 , 0
  4721.5     .05       0  4996.8     .05       0  5000.8     .05       0
  5100.1     .12       0    5147     .05       0  5316.8     .12       0
Bank Sta=4996.8,5000.8
XS Rating Curve= 0 ,0
Exp/Cntr=0.3,0.1

Type RM Length L Ch R = 1 ,16000   ,500,500,500
BEGIN DESCRIPTION:
MAGILL CREEK 32.0
END DESCRIPTION:
XS GIS Cut Line= 3
      2787305.69     10290253.11      2787051.45     10289996.68
      2786855.69     10289803.12
#Sta/Elev= 30
  4638.9 1382.22  4667.2 1381.78  4709.6 1379.72    4745 1376.62  4780.3 1372.28
  4822.7 1368.08  4886.4 1362.38  4893.4 1360.81  4914.7 1358.12    4943 1358.55
  4978.3 1357.88  4992.4 1355.34    4999 1353.25  5004.6 1352.85  5004.9 1352.35
  5008.4 1352.35  5008.6 1352.85  5020.8 1353.86  5027.8 1355.95  5034.9 1355.98
    5042 1357.52  5098.5 1363.05  5176.3 1372.89  5197.5 1374.86  5204.6 1376.26
  5211.7 1376.38  5261.2 1382.38  5268.2 1382.69  5271.8 1384.22  5275.3 1384.22
#Mann= 3 ,-1 , 0
  4638.9     .05       0  5004.6     .05       0  5008.6     .05       0
Bank Sta=5004.6,5008.6
XS Rating Curve= 0 ,0
Exp/Cntr=0.3,0.1

Type RM Length L Ch R = 1 ,15500   ,500,500,500
BEGIN DESCRIPTION:
MAGILL CREEK 31.0
END DESCRIPTION:
XS GIS Cut Line= 3
      2787555.68     10290203.09       2787473.1     10289814.87
      2787405.69     10289603.14
#Sta/Elev= 30
  4603.1 1374.08  4622.8 1373.29  4627.9 1373.76  4734.8 1367.87  4807.6 1364.37
    4828 1362.55  4848.4 1361.95  4879.1 1360.04  4889.3 1358.51  4899.6 1358.07
  4959.7 1352.71  4964.8  1351.8  4979.4 1347.12  4979.6 1346.62  4983.1 1346.62
  4983.4 1347.12  5003.5 1347.98  5007.5 1350.19  5012.8 1350.19  5022.8 1351.92
  5064.8 1353.95  5077.2 1355.84  5096.3 1357.71  5104.2  1359.6  5148.8 1365.54
  5180.6 1368.59  5206.1 1369.41  5211.7 1370.23    5221 1370.51  5222.2 1370.51
#Mann= 6 ,-1 , 0
  4603.1     .05       0  4734.8     .12       0  4979.4     .07       0
  4983.4     .12       0  5180.6     .05       0    5221     .12       0
Bank Sta=4979.4,4983.4
XS Rating Curve= 0 ,0
Exp/Cntr=0.3,0.1

Type RM Length L Ch R = 1 ,15000   ,500,500,500
BEGIN DESCRIPTION:
MAGILL CREEK 30.0
END DESCRIPTION:
XS GIS Cut Line= 3
      2788305.71     10290003.13      2787927.69     10289616.81
       2787555.7     10289403.12
#Sta/Elev= 30
  4459.5 1420.42  4478.6  1418.4  4487.7 1416.34  4494.9 1416.28    4516 1410.51
  4551.5  1404.1  4579.8  1402.4  4600.9 1398.13  4681.1 1387.03  4721.2 1382.83
  4756.5 1376.03  4777.8 1370.45  4784.8 1371.36  4791.9 1368.74  4798.9 1368.64
  4820.2  1364.5  4884.4 1355.56  4926.2 1351.85  4968.1 1345.77  4975.8 1343.32
  4987.9 1342.65  4988.2 1342.15    4992 1342.65  5016.1 1345.47  5071.5 1347.64
  5127.3 1352.35  5165.7 1354.54  5238.4 1359.45  5378.9 1367.42    5429  1369.7
#Mann= 12 ,-1 , 0
  4459.5     .05       0  4478.6     .12       0  4681.1     .05       0
  4884.4     .12       0  4968.1     .05       0  4987.9     .05       0
    4992     .05       0  5016.1     .12       0  5127.3     .05       0
  5165.7     .12       0  5238.4     .05       0  5378.9     .12       0
Bank Sta=4987.9,4992
XS Rating Curve= 0 ,0
Exp/Cntr=0.3,0.1

Type RM Length L Ch R = 1 ,14500   ,500,500,500
BEGIN DESCRIPTION:
MAGILL CREEK 29.0
END DESCRIPTION:
XS GIS Cut Line= 3
      2788305.69     10289503.12      2788186.54     10289240.05
      2787855.69     10289203.11
#Sta/Elev= 30
  4711.2 1375.86  4734.3 1373.25  4748.6 1371.94  4771.7 1366.36  4788.1 1364.41
  4817.9 1358.94    4841  1352.8  4846.5 1352.84  4875.9 1345.59  4884.2 1345.02
  4892.7 1345.92  4898.2 1343.92  4915.8 1342.34  4921.3 1340.29  4930.8 1338.45
  4938.9 1338.25  4944.4 1336.66  4952.7  1337.3    4983 1336.31  4983.3 1335.81
  4987.2 1336.31  5002.9 1336.54  5016.7 1340.87  5051.2  1344.2  5061.2  1344.3
  5112.1 1351.11  5131.7 1352.59    5191 1354.03  5327.2 1359.47  5332.9  1359.5
#Mann= 7 ,-1 , 0
  4711.2     .05       0  4734.3     .12       0  4884.2     .05       0
    4983     .05       0  4987.2     .05       0    5191     .12       0
  5327.2     .05       0
Bank Sta=4983,4987.2
XS Rating Curve= 0 ,0
Exp/Cntr=0.3,0.1

Type RM Length L Ch R = 1 ,14000   ,500,500,500
BEGIN DESCRIPTION:
MAGILL CREEK 28.0
END DESCRIPTION:
XS GIS Cut Line= 3
       2788455.7     10289003.14      2788333.48     10288765.41
       2788155.7     10288553.13
#Sta/Elev= 30
  4732.7 1350.91  4785.4 1349.79  4813.2  1346.5  4829.7 1347.17  4835.3 1344.21
  4874.1 1342.13  4879.7 1340.17  4890.1 1339.97  4901.9 1336.24  4918.4 1333.86
  4924.1 1330.76  4960.6 1327.09  4960.9 1326.59    4965 1327.09    4985 1328.15
  5002.2 1327.31  5014.7 1328.33  5021.2 1330.95  5035.6 1332.67  5049.9 1332.31
  5056.4 1333.69  5078.5 1333.75  5127.9 1337.14  5148.8 1342.84  5156.6 1343.29
  5163.1 1346.13  5170.9 1345.88  5212.5 1353.86  5256.8 1359.66  5276.9 1360.81
#Mann= 4 ,-1 , 0
  4732.7     .12       0  4960.6     .07       0    4965     .12       0
  5256.8     .05       0
Bank Sta=4960.6,4965
XS Rating Curve= 0 ,0
Exp/Cntr=0.3,0.1

Type RM Length L Ch R = 1 ,13500   ,500,500,500
BEGIN DESCRIPTION:
MAGILL CREEK 27.0
END DESCRIPTION:
XS GIS Cut Line= 3
       2789055.7     10288903.12       2788647.8     10288633.42
      2788455.69     10288303.12
#Sta/Elev= 30
    4511 1394.67  4533.6 1393.25  4581.6 1377.59    4613 1366.53  4684.1 1343.19
  4705.1 1341.34  4750.3 1345.32  4770.1 1342.89  4792.4 1336.84  4807.5 1339.84
  4813.4 1336.11  4849.6 1327.39  4891.8 1325.55    4988 1321.55    4994 1319.26
  5007.9 1318.91  5008.2 1318.41  5012.4 1318.91  5074.7 1324.51  5090.4 1330.05
  5111.9 1333.94  5117.7 1332.04  5185.5 1338.21    5251 1349.74  5278.3 1358.48
  5309.7 1364.57  5315.5 1368.35    5337 1374.69  5346.8 1375.14  5382.1 1369.17
#Mann= 8 ,-1 , 0
    4511     .12       0  4581.6     .05       0    4613     .12       0
  4770.1     .05       0  4891.8     .12       0  5007.9     .07       0
  5012.4     .12       0  5346.8     .05       0
Bank Sta=5007.9,5012.4
XS Rating Curve= 0 ,0
Exp/Cntr=0.3,0.1

Type RM Length L Ch R = 1 ,13000   ,500,500,500
BEGIN DESCRIPTION:
MAGILL CREEK 26.0
END DESCRIPTION:
XS GIS Cut Line= 3
      2789155.69     10288503.12      2789037.62     10288422.62
      2788855.65      10288353.1
#Sta/Elev= 30
  4857.1 1347.14  4860.1 1347.14  4864.6  1344.5  4879.5 1342.29  4885.6 1341.94
  4896.9 1339.86  4906.5 1337.86  4929.7 1330.49  4936.4 1329.15  4951.3 1324.18
  4957.4 1323.25  4972.3 1317.74  4978.3 1316.55  4987.2 1312.46  4995.9 1310.04
  4996.2 1309.54  5000.1 1309.54  5000.4 1310.04  5003.7 1310.04  5015.4  1311.6
  5023.5 1313.98  5045.5 1318.08  5055.6 1317.49    5077 1321.98  5087.7 1323.05
  5105.7 1326.33  5141.2 1329.94    5155 1330.31  5185.1 1334.29  5194.8 1333.91
#Mann= 5 ,-1 , 0
  4857.1     .05       0  4896.9     .12       0  4995.9     .07       0
  5000.4     .12       0  5105.7     .05       0
Bank Sta=4995.9,5000.4
XS Rating Curve= 0 ,0
Exp/Cntr=0.3,0.1

Type RM Length L Ch R = 1 ,12500   ,500,500,500
BEGIN DESCRIPTION:
MAGILL CREEK 25.0
END DESCRIPTION:
XS GIS Cut Line= 3
      2789255.66     10287953.12      2789012.14     10287992.59
      2788655.69     10288253.11
#Sta/Elev= 30
  4753.3 1347.64  4781.6 1345.27  4786.6  1342.7  4814.1 1337.25  4843.2 1327.84
  4854.6 1321.44  4876.2 1314.01  4895.1  1308.1  4904.8 1307.67  4915.4  1303.6
    4966 1303.39  4971.5 1301.39    4984 1300.92  4984.3 1300.42  4988.6 1300.92
  5005.6 1300.93  5011.8 1303.05  5041.1 1305.06    5062 1310.29  5097.5 1313.87
  5107.7 1316.23  5162.3 1321.12  5212.5 1321.59  5272.6 1325.87    5384 1335.28
  5404.8 1342.42  5413.3 1347.43  5419.5  1346.5  5430.1 1349.33  5441.5 1353.06
#Mann= 7 ,-1 , 0
  4753.3     .12       0  4876.2     .05       0    4984     .05       0
  4988.6     .05       0  5107.7     .12       0  5272.6     .05       0
  5430.1     .12       0
Bank Sta=4984,4988.6
XS Rating Curve= 0 ,0
Exp/Cntr=0.3,0.1

Type RM Length L Ch R = 1 ,12000   ,500,500,500
BEGIN DESCRIPTION:
MAGILL CREEK 24.0
END DESCRIPTION:
XS GIS Cut Line= 3
      2789005.64     10287653.12      2788623.83     10287691.14
      2788555.68     10287953.12
#Sta/Elev= 30
  4616.3 1328.61  4656.5 1325.85  4676.6 1326.27  4735.4 1324.17  4746.9 1323.79
    4757 1322.24  4764.8 1319.04  4807.2 1309.52  4817.2  1308.5  4857.4 1308.14
  4887.6 1303.86  4907.7 1305.93  4947.9 1301.37  4971.2 1295.83  4985.8 1293.52
  4986.1 1293.02  4990.4 1293.52  5003.6    1294  5009.9 1295.21  5013.3 1296.62
  5043.4 1301.87  5055.5 1304.71  5084.7 1308.42  5090.9  1310.1  5113.6 1313.09
    5157 1319.73  5212.5 1325.07    5253 1330.35  5268.1 1334.82  5270.7 1334.82
#Mann= 6 ,-1 , 0
  4616.3     .05       0  4735.4     .12       0  4985.8     .07       0
  4990.4     .12       0  5013.3     .05       0  5113.6     .12       0
Bank Sta=4985.8,4990.4
XS Rating Curve= 0 ,0
Exp/Cntr=0.3,0.1

Type RM Length L Ch R = 1 ,11500   ,500,500,500
BEGIN DESCRIPTION:
MAGILL CREEK 23.0
END DESCRIPTION:
XS GIS Cut Line= 3
      2788805.71     10287353.12      2788381.25     10287271.67
      2787905.68     10287503.11
#Sta/Elev= 30
  4567.8  1312.6  4697.8 1306.45  4791.8  1303.5  4858.9 1298.43  4924.2 1297.74
  4934.4  1300.7  4944.6 1300.26  4954.8 1297.67  4962.8  1294.1  4967.9 1293.71
    4983 1287.56  4983.3 1287.06  4987.7 1287.56  5021.8 1290.35  5058.3 1296.14
  5063.9 1298.18  5139.6 1299.95  5176.6 1306.79  5193.6 1308.06  5199.2 1310.67
  5206.4 1311.45  5216.2 1310.28  5221.7 1311.69  5286.7 1314.17  5306.4 1315.52
  5317.6  1317.7  5373.2 1321.75  5492.3 1339.65  5528.2 1342.55  5528.9 1342.55
#Mann= 6 ,-1 , 0
  4567.8     .05       0    4983     .05       0  4987.7     .05       0
  5021.8     .12       0  5286.7     .05       0  5528.2     .12       0
Bank Sta=4983,4987.7
XS Rating Curve= 0 ,0
Exp/Cntr=0.3,0.1

Type RM Length L Ch R = 1 ,11000   ,500,500,500
BEGIN DESCRIPTION:
MAGILL CREEK 22.0
END DESCRIPTION:
XS GIS Cut Line= 3
       2788955.7     10287253.12      2788560.16     10286849.95
      2788505.69     10286353.13
#Sta/Elev= 30
  4435.2  1330.7  4438.7  1330.7  4442.3 1328.26  4456.4 1327.13  4484.7 1329.05
  4504.6 1327.57  4527.2 1323.16  4541.3  1324.7  4562.4 1322.37  4569.6 1318.84
  4576.6  1312.8  4583.7 1310.84  4590.7 1305.82  4597.9 1304.34  4668.6 1299.62
  4802.9 1294.42    4810 1292.59  4838.3 1292.61  4944.3 1284.85  4984.1 1279.16
  4984.5 1278.66  4989.5 1279.16  5047.1 1283.56  5101.2 1282.62  5117.5 1281.45
  5137.7  1286.2  5248.3 1298.65  5363.1 1308.94    5497 1323.54  5499.8 1323.59
#Mann= 6 ,-1 , 0
  4435.2     .12       0  4504.6     .05       0  4984.1     .05       0
  4989.5     .05       0  5101.2     .12       0    5497     .05       0
Bank Sta=4984.1,4989.5
XS Rating Curve= 0 ,0
Exp/Cntr=0.3,0.1

Type RM Length L Ch R = 1 ,10500   ,500,500,500
BEGIN DESCRIPTION:
MAGILL CREEK 21.0
END DESCRIPTION:
XS GIS Cut Line= 3
       2789255.7     10287003.13      2788987.05     10286614.93
      2788805.72     10286403.15
#Sta/Elev= 30
  4527.9    1330  4535.4 1330.39  4541.4 1325.04  4550.2 1323.23  4556.3 1318.99
  4571.2 1317.16  4592.1 1310.84  4600.1  1310.6    4607 1310.55  4613.1 1306.79
  4621.9 1305.77  4627.9 1302.21  4636.7 1302.69  4642.8 1299.03  4649.5 1297.84
  4750.2 1290.82  4786.1 1282.36  4857.7 1285.61  4929.3 1282.44  4959.1 1279.97
  4973.9 1274.59  4995.3 1270.93  4995.8 1270.43  5000.8 1270.93  5037.9 1278.21
  5087.3 1282.72  5115.7 1290.12  5158.7 1299.44  5203.1 1304.69  5278.8 1313.65
#Mann= 6 ,-1 , 0
  4527.9     .05       0  4600.1     .12       0  4995.3     .07       0
  5000.8     .12       0  5115.7     .05       0  5203.1     .12       0
Bank Sta=4995.3,5000.8
XS Rating Curve= 0 ,0
Exp/Cntr=0.3,0.1

Type RM Length L Ch R = 1 ,10000   ,500,500,500
BEGIN DESCRIPTION:
MAGILL CREEK 20.0
END DESCRIPTION:
XS GIS Cut Line= 3
      2789555.68     10286903.08      2789465.52     10286493.79
       2789405.7     10286303.15
#Sta/Elev= 30
  4580.9 1305.13  4583.4 1305.13  4600.2 1300.12  4605.3 1299.88  4611.6 1297.24
  4642.3 1295.82  4683.8 1292.08  4726.8 1289.25  4747.2 1288.31  4785.3 1286.72
  4806.1 1286.92  4828.3  1286.1  4877.8 1284.22  4918.8 1280.53  4959.7 1275.42
    4970 1275.31  4980.7 1270.83    4995 1266.61  4995.4 1266.11  5000.1 1266.11
  5000.5 1266.61  5074.1 1273.12    5095 1277.27  5118.8 1279.81    5137 1284.45
    5146  1287.6  5168.4 1291.83  5183.6 1293.58  5197.2 1297.25  5199.8 1297.25
#Mann= 7 ,-1 , 0
  4580.9     .05       0  4683.8     .12       0  4726.8     .05       0
  4747.2     .12       0  4828.3     .05       0    4995     .05       0
  5000.5     .05       0
Bank Sta=4995,5000.5
XS Rating Curve= 0 ,0
Exp/Cntr=0.3,0.1

Type RM Length L Ch R = 1 ,9500    ,500,500,500
BEGIN DESCRIPTION:
MAGILL CREEK 19.0
END DESCRIPTION:
XS GIS Cut Line= 3
      2789905.69     10286553.13      2789826.51     10286167.06
      2789605.68     10286103.11
#Sta/Elev= 30
  4605.9 1285.42  4646.7 1283.51  4678.8 1283.49  4731.9 1283.38  4769.2 1281.42
  4789.7 1281.81  4832.7 1279.79  4871.3 1276.92  4881.1 1275.46    4902 1272.01
  4922.4 1269.79  4933.6 1266.65  4942.8 1265.93  4963.2 1261.49  4978.9 1260.19
    4984  1258.5  4996.7 1258.02  4997.1 1257.52  5001.8 1257.52  5002.3 1258.02
  5011.3 1258.55  5025.2 1264.03  5042.5 1273.24  5073.7 1278.55  5086.5  1279.8
  5167.4 1286.18  5174.3  1287.4  5179.5 1287.28  5198.7 1289.03  5229.9 1292.73
#Mann= 7 ,-1 , 0
  4605.9     .12       0  4678.8     .05       0  4881.1     .12       0
  4996.7     .07       0  5002.3     .12       0  5025.2     .05       0
  5086.5     .12       0
Bank Sta=4996.7,5002.3
XS Rating Curve= 0 ,0
Exp/Cntr=0.3,0.1

Type RM Length L Ch R = 1 ,9000    ,500,500,500
BEGIN DESCRIPTION:
MAGILL CREEK 18.0
END DESCRIPTION:
XS GIS Cut Line= 3
      2790305.65      10285853.1       2790059.1     10285763.88
      2789555.71     10285403.13
#Sta/Elev= 30
  4737.8 1275.67  4783.7 1273.27  4833.5 1272.71  4886.6 1269.65  4939.8 1263.25
  4950.5 1261.13    4957 1257.75  4962.3 1258.14  4996.2 1253.47  4996.7 1252.97
  5002.1 1253.47    5031 1257.74  5060.5 1264.43  5080.5 1266.11  5089.9 1268.39
  5125.6 1270.91  5172.5 1268.92  5217.7 1267.95  5290.4 1272.43  5339.3 1276.42
  5357.1 1279.66  5368.8    1281  5374.9 1283.31  5410.5 1289.63  5469.8 1297.81
  5496.5 1302.33  5540.7 1306.96  5553.4 1310.03  5576.3 1312.37  5619.3 1320.65
#Mann= 9 ,-1 , 0
  4737.8     .12       0  4996.2     .07       0  5002.1     .12       0
  5080.5     .05       0  5172.5     .12       0  5290.4     .05       0
  5357.1     .12       0  5469.8     .05       0  5553.4     .12       0
Bank Sta=4996.2,5002.1
XS Rating Curve= 0 ,0
Exp/Cntr=0.3,0.1

Type RM Length L Ch R = 1 ,8500    ,500,500,500
BEGIN DESCRIPTION:
MAGILL CREEK 17.0
END DESCRIPTION:
XS GIS Cut Line= 3
      2790405.67      10285503.1      2790139.83     10285272.69
      2789955.73     10285203.13
#Sta/Elev= 30
  4648.2 1274.89  4661.9 1274.22  4712.3  1268.5  4733.2 1266.85  4754.1 1262.79
  4761.7 1262.26  4811.1 1261.25  4825.3 1260.17  4888.9  1259.8    4903 1259.15
  4952.5 1253.92  4988.7    1252  4996.4 1250.52  4996.9 1250.02  5001.9 1250.02
  5002.4 1250.52  5004.9 1250.52  5011.4 1258.75  5016.7 1257.57  5025.8 1262.92
  5036.2 1264.88  5066.4 1267.61  5071.7 1267.46  5111.3 1272.22  5128.9 1273.16
  5135.9  1274.1  5156.9 1275.22  5181.8 1278.01  5187.1 1277.52  5196.8 1278.15
#Mann= 6 ,-1 , 0
  4648.2     .05       0    4903     .12       0  4996.4     .07       0
  5002.4     .12       0  5128.9     .05       0  5135.9     .12       0
Bank Sta=4996.4,5002.4
XS Rating Curve= 0 ,0
Exp/Cntr=0.3,0.1

Type RM Length L Ch R = 1 ,8000    ,500,500,500
BEGIN DESCRIPTION:
MAGILL CREEK 16.0
END DESCRIPTION:
XS GIS Cut Line= 3
      2790605.68     10285403.11      2790527.13     10284993.78
      2790155.69     10284653.12
#Sta/Elev= 30
  4583.2 1270.75  4765.2 1268.94  4847.9 1264.95  4874.2 1262.49  4919.2 1255.29
  4926.2 1253.71  4931.3 1250.47  4970.1 1247.64  4978.2 1248.27  4994.8 1247.09
  4995.3 1246.59  5000.8 1247.09  5008.6 1247.37  5022.7    1251  5029.5 1251.16
  5065.3 1257.09  5107.8 1260.31  5157.2 1266.75  5164.6 1266.04  5171.4 1268.05
  5185.5 1267.62  5206.5 1270.29  5270.6 1274.56  5334.1 1281.72  5348.3 1281.92
  5362.5 1285.19  5390.9 1288.75  5411.8 1294.48    5476  1304.1    5504 1310.09
#Mann= 3 ,-1 , 0
  4583.2     .05       0  4994.8     .05       0  5000.8     .05       0
Bank Sta=4994.8,5000.8
XS Rating Curve= 0 ,0
Exp/Cntr=0.3,0.1

Type RM Length L Ch R = 1 ,7500    ,500,500,500
BEGIN DESCRIPTION:
MAGILL CREEK 15.0
END DESCRIPTION:
XS GIS Cut Line= 3
      2791355.68     10285253.11      2790973.01     10284868.57
       2790755.7     10284653.13
#Sta/Elev= 30
  4457.5 1265.85  4620.1 1261.51  4761.6 1261.47    4811  1263.1  4874.7 1263.12
    4903 1260.68  4938.3 1259.67  4952.5 1253.45  4959.5 1248.71  4966.6 1249.09
  4973.7 1244.56  4980.7 1244.99  4996.9 1243.46  4997.4 1242.96    5003 1243.46
  5009.1 1243.69  5015.1 1245.29  5023.2  1245.6  5030.2  1247.2  5058.5 1248.72
  5065.6 1248.27  5093.9 1252.26    5101 1254.35  5108.1 1254.49  5136.3 1262.15
  5164.6 1265.58    5200 1266.37  5207.1 1267.85  5287.6 1268.52    5306 1268.84
#Mann= 5 ,-1 , 0
  4457.5     .05       0  4996.9     .03       0    5003     .05       0
  5015.1     .12       0  5287.6     .05       0
Bank Sta=4996.9,5003
XS Rating Curve= 0 ,0
Exp/Cntr=0.3,0.1

Type RM Length L Ch R = 1 ,7000    ,500,500,500
BEGIN DESCRIPTION:
MAGILL CREEK 14.0
END DESCRIPTION:
XS GIS Cut Line= 3
      2791505.68     10285103.12      2791429.34     10284692.55
      2791055.71     10284503.13
#Sta/Elev= 30
  4582.4 1263.26  4661.6 1260.14  4765.5 1257.69    4796  1255.7  4806.2 1256.91
  4836.7 1258.22  4918.1  1254.7  4940.7 1254.25  4948.6 1253.17  4968.9 1247.11
  4993.5  1241.1  4994.1 1239.86  4994.6 1239.36  4999.7 1239.36  5000.2 1239.86
  5009.8 1240.05  5015.4 1241.12  5026.4 1241.93    5032 1243.43  5054.3 1245.04
  5060.2    1247  5076.6 1249.61  5149.8 1252.97  5172.3 1253.36  5254.7 1257.65
  5315.9 1259.88  5329.2 1260.92  5351.7 1261.85  5371.7 1261.88  5418.9 1262.79
#Mann= 4 ,-1 , 0
  4582.4     .05       0  4994.1     .03       0  5000.2     .05       0
  5371.7     .12       0
Bank Sta=4994.1,5000.2
XS Rating Curve= 0 ,0
Exp/Cntr=0.3,0.1

Type RM Length L Ch R = 1 ,6500    ,500,500,500
BEGIN DESCRIPTION:
MAGILL CREEK 13.0
END DESCRIPTION:
XS GIS Cut Line= 3
       2792005.7     10284903.16      2791894.31     10284512.73
      2792155.67     10284003.15
#Sta/Elev= 30
    4594 1257.44  4656.4  1255.3  4790.5 1244.97    4854 1244.13  4868.5 1242.42
  4885.2 1243.92  4907.5 1243.47  4941.4 1241.87  4989.2 1238.37  4994.1 1237.15
  4994.6 1236.65  5000.3 1237.15  5015.2 1237.22  5031.8 1241.29  5037.4 1240.41
    5067 1247.69  5224.3 1248.75  5259.3 1247.16  5269.3 1248.66  5306.1 1246.79
  5314.3 1246.43  5320.3 1244.63  5325.9 1245.17  5336.7 1241.59  5348.1 1240.77
  5364.7 1245.46  5370.4 1250.31  5386.9 1254.44  5453.5 1256.47  5572.7 1262.88
#Mann= 4 ,-1 , 0
    4594     .05       0  4994.1     .05       0  5000.3     .05       0
  5306.1     .12       0
Bank Sta=4994.1,5000.3
XS Rating Curve= 0 ,0
Exp/Cntr=0.3,0.1

Type RM Length L Ch R = 1 ,6000    ,500,500,500
BEGIN DESCRIPTION:
MAGILL CREEK 12.0
END DESCRIPTION:
XS GIS Cut Line= 3
      2792305.68     10284853.13      2792362.14      10284605.9
      2792305.69     10284103.16
#Sta/Elev= 30
  4746.4 1253.41    4808 1249.77  4869.5 1247.67  4904.5 1247.19  4920.8 1245.23
  4947.5 1240.24  4961.8 1239.89  4982.3 1237.68  4986.5  1233.2    4987  1232.7
    4994  1232.7  4994.5  1233.2  4995.6  1235.5  4998.9 1233.37  5003.9 1233.37
  5015.5  1234.8  5022.9 1236.61  5063.2 1238.02  5093.4 1237.64  5105.5 1239.22
  5123.6  1245.6  5133.6 1246.67  5153.7 1247.13  5242.8 1246.72  5324.8 1249.75
    5355  1251.7  5375.8 1251.86  5445.6 1254.62  5474.5 1256.35  5505.9 1257.48
#Mann= 5 ,-1 , 0
  4746.4     .05       0  4986.5     .03       0  4994.5     .05       0
  5242.8     .12       0  5474.5     .05       0
Bank Sta=4986.5,4994.5
XS Rating Curve= 0 ,0
Exp/Cntr=0.3,0.1

Type RM Length L Ch R = 1 ,5500    ,500,500,500
BEGIN DESCRIPTION:
MAGILL CREEK 11.0
END DESCRIPTION:
XS GIS Cut Line= 3
      2792605.69     10284903.11      2792793.53     10284498.92
      2792755.68     10284153.09
#Sta/Elev= 30
  4554.3 1253.19  4614.3 1251.17  4697.6  1247.2  4808.4 1243.68  4922.9 1242.02
  4940.2 1240.36  4945.8 1237.94  4951.3 1238.73  4962.3 1236.88  4968.7 1233.98
  4974.2 1236.15  4984.4 1232.04  4992.6 1230.52  4993.1 1230.02  5000.1 1230.02
  5000.6 1230.52  5015.9 1233.12    5036 1235.08  5053.9 1237.89  5076.3 1240.01
  5096.4 1240.95  5114.8 1240.86  5126.6 1242.48  5146.7  1243.8  5186.9 1244.71
    5206  1246.5  5237.2 1247.86  5297.2 1251.98  5317.7 1252.44  5347.9 1254.68
#Mann= 4 ,-1 , 0
  4554.3     .05       0  4992.6     .03       0  5000.6     .05       0
  5053.9     .12       0
Bank Sta=4992.6,5000.6
XS Rating Curve= 0 ,0
Exp/Cntr=0.3,0.1

Type RM Length L Ch R = 1 ,5000    ,500,500,500
BEGIN DESCRIPTION:
MAGILL CREEK 10.0
END DESCRIPTION:
XS GIS Cut Line= 3
      2792905.66     10284903.14      2793254.39     10284485.88
       2793355.7     10284303.08
#Sta/Elev= 30
  4456.2 1248.25  4498.5 1245.67  4590.9 1241.68  4626.1 1237.41  4662.5 1235.05
  4804.4  1233.5  4882.4 1234.81    4889  1234.1  4911.1 1234.85  4917.6 1234.08
  4925.4 1234.87  4931.9 1233.26  4946.2 1233.46  4952.7  1232.1  4974.8 1230.74
  4994.5  1227.7    4995  1227.2  5002.6  1227.7  5010.9 1228.06  5016.7 1230.08
  5022.8    1231  5032.7 1233.65  5038.4  1236.5  5040.9 1237.04  5054.4 1240.33
  5060.3 1242.73  5076.2 1246.17  5132.5 1250.06    5188 1254.16    5209 1256.14
#Mann= 7 ,-1 , 0
  4456.2     .05       0  4994.5     .03       0  5002.6     .05       0
  5022.8     .12       0  5040.9     .05       0  5132.5     .12       0
    5188     .05       0
Bank Sta=4994.5,5002.6
XS Rating Curve= 0 ,0
Exp/Cntr=0.3,0.1

Type RM Length L Ch R = 1 ,4500    ,500,500,500
BEGIN DESCRIPTION:
MAGILL CREEK 9.0
END DESCRIPTION:
XS GIS Cut Line= 3
      2793505.69     10285253.15       2793398.9     10284866.63
      2793505.68     10284353.12
#Sta/Elev= 30
    4599 1260.54  4621.4 1257.96  4690.1 1252.55  4729.6 1247.77  4835.1  1239.7
  4858.4 1238.94  4877.3 1236.66  4882.5 1237.33  4899.9 1235.13  4910.3 1232.53
    4922 1227.96    4931  1229.2  4951.2 1227.91  4956.4 1228.59  4982.9 1225.76
  4995.2 1222.63  4995.7 1222.13  5003.3 1222.63  5008.7 1225.07  5034.2  1227.3
  5053.7 1233.42  5058.8  1232.9  5064.9 1235.25  5075.1 1236.31  5115.9 1237.66
  5153.9 1240.36  5254.1 1240.51  5381.5  1244.1  5432.6 1247.11  5524.5 1254.59
#Mann= 4 ,-1 , 0
    4599     .12       0  4835.1     .05       0  4995.2     .05       0
  5003.3     .05       0
Bank Sta=4995.2,5003.3
XS Rating Curve= 0 ,0
Exp/Cntr=0.3,0.1

Type RM Length L Ch R = 1 ,4000    ,500,500,500
BEGIN DESCRIPTION:
MAGILL CREEK 8.0
END DESCRIPTION:
XS GIS Cut Line= 3
      2793855.69     10285153.08      2793891.55       10284918.
      2793555.71     10284403.15
#Sta/Elev= 30
  4762.2 1254.41  4772.3  1254.3  4791.4 1251.96  4796.4 1251.98    4860 1242.11
    4865 1242.16  4893.7 1238.97  4923.5 1234.17  4928.5 1234.96  4934.1 1232.75
  4964.5 1227.33  4974.6 1223.01  4992.9 1219.93  4993.4 1219.43  5000.7 1219.43
  5001.2 1219.93  5006.7 1220.14  5015.8 1222.21  5021.8 1222.15  5036.9 1229.42
  5052.1 1232.56  5330.6 1238.87    5405 1240.01  5498.6 1243.29    5530 1245.07
  5555.9 1246.15    5565 1247.14    5571 1246.83  5601.2 1249.79  5614.7 1250.47
#Mann= 5 ,-1 , 0
  4762.2     .05       0  4992.9     .05       0  5001.2     .05       0
  5330.6     .12       0    5530     .05       0
Bank Sta=4992.9,5001.2
XS Rating Curve= 0 ,0
Exp/Cntr=0.3,0.1

Type RM Length L Ch R = 1 ,3500    ,500,500,500
BEGIN DESCRIPTION:
MAGILL CREEK 7.0
END DESCRIPTION:
XS GIS Cut Line= 3
      2794155.68     10285203.12      2794359.91     10284787.71
      2794305.68     10284453.07
#Sta/Elev= 30
  4537.1 1245.13    4568 1244.29  4618.6 1239.88  4635.5  1240.9  4663.5    1238
  4680.4 1238.23    4686 1236.45  4702.9 1237.57  4708.5 1233.94  4725.4 1237.41
  4730.9 1232.76  4747.8 1238.88  4753.4 1237.62    4760 1238.91  4820.8 1233.25
  4860.2 1233.78  4905.3 1229.89  4949.4 1228.18  4955.7  1224.7  4961.3 1226.74
  4978.2 1217.83  4983.8 1218.65  4989.7 1216.37  4990.2 1215.87  4998.2 1216.37
  5075.6 1224.31    5106 1233.23  5194.3 1236.49  5290.5 1239.25    5339 1240.78
#Mann= 6 ,-1 , 0
  4537.1     .05       0  4905.3     .12       0  4989.7     .07       0
  4998.2     .12       0  5194.3     .05       0  5290.5     .12       0
Bank Sta=4989.7,4998.2
XS Rating Curve= 0 ,0
Exp/Cntr=0.3,0.1

Type RM Length L Ch R = 1 ,3000    ,500,500,500
BEGIN DESCRIPTION:
MAGILL CREEK 6.0
END DESCRIPTION:
XS GIS Cut Line= 3
       2794655.7     10285103.09      2794849.94     10284862.25
      2794805.68     10284503.07
#Sta/Elev= 30
  4690.6 1235.24  4754.8 1233.88  4896.1  1229.3  4939.3 1228.55  4947.2 1226.96
  4953.7 1227.28  4960.4    1226  4968.1  1222.2  4974.5 1223.61  4982.4 1216.14
  4988.9 1215.56  4991.9 1212.93  4992.4 1212.43    5000 1212.43  5000.5 1212.93
  5019.3 1213.46  5033.9 1216.28  5039.4 1217.48  5069.7 1219.67    5120 1224.52
  5150.3 1227.54  5156.4 1229.39  5170.4 1230.22  5200.6 1230.25  5237.6 1231.48
    5251 1231.17  5311.5 1232.55  5318.7  1232.1  5341.7 1233.98  5361.9 1234.09
#Mann= 4 ,-1 , 0
  4690.6     .05       0  4991.9     .05       0  5000.5     .05       0
  5033.9     .12       0
Bank Sta=4991.9,5000.5
XS Rating Curve= 0 ,0
Exp/Cntr=0.3,0.1

Type RM Length L Ch R = 1 ,2500    ,500,500,500
BEGIN DESCRIPTION:
MAGILL CREEK 5.0
END DESCRIPTION:
XS GIS Cut Line= 3
      2795305.68     10285303.11      2795335.24     10284914.23
      2795455.68     10284403.13
#Sta/Elev= 30
    4610 1231.04  4710.3 1229.84  4740.4 1230.47  4750.4 1229.74  4770.5  1230.5
  4860.7 1227.53  4890.8 1224.81  4900.8 1222.59  4930.9 1211.13    4961 1211.98
  4981.1 1211.51  4993.4 1210.34  4993.9 1209.84  5002.7 1210.34  5011.4 1210.84
  5042.2 1217.21  5062.5 1218.29  5067.6 1217.32  5074.4 1218.52  5093.6 1218.88
  5124.4 1223.19    5145 1224.82  5268.3 1229.82    5332 1233.62  5365.4 1237.29
  5369.2 1238.01  5374.3 1237.67  5411.5 1242.37  5465.3 1246.32  5525.1 1251.01
#Mann= 6 ,-1 , 0
    4610     .05       0  4993.4     .05       0  5002.7     .05       0
  5074.4     .12       0  5365.4     .05       0  5465.3     .12       0
Bank Sta=4993.4,5002.7
XS Rating Curve= 0 ,0
Exp/Cntr=0.3,0.1

Type RM Length L Ch R = 1 ,2000    ,500,500,500
BEGIN DESCRIPTION:
MAGILL CREEK 4.0
END DESCRIPTION:
XS GIS Cut Line= 3
       2795455.7      10285403.1      2795822.14     10284980.69
      2795905.69     10284653.08
#Sta/Elev= 30
  4440.8 1232.14  4582.8 1226.56    4710 1223.73  4916.1 1221.46  4943.8 1219.29
  4965.5 1212.03  4972.1 1211.59  4994.1 1206.62  4994.6 1206.12  5003.6 1206.62
  5009.8 1207.28  5039.3 1212.31  5059.4 1213.67  5069.7 1211.81    5075  1213.3
  5080.1 1217.89  5100.7 1220.38  5151.6 1220.89  5156.7 1223.08  5172.9 1223.54
  5192.4 1221.04  5197.6 1223.57  5201.7 1223.25  5224.5 1222.85  5238.5 1225.08
  5274.2 1225.17  5312.9 1227.94  5320.2 1227.87  5335.5 1235.12  5338.1 1235.12
#Mann= 6 ,-1 , 0
  4440.8     .05       0  4994.1     .03       0  5003.6     .05       0
  5009.8     .12       0  5201.7     .05       0  5312.9     .12       0
Bank Sta=4994.1,5003.6
XS Rating Curve= 0 ,0
Exp/Cntr=0.3,0.1

Type RM Length L Ch R = 1 ,1500    ,500,500,500
BEGIN DESCRIPTION:
MAGILL CREEK 3.0
END DESCRIPTION:
XS GIS Cut Line= 3
      2795705.72     10285653.08      2796229.99     10285263.78
       2796455.7     10284903.08
#Sta/Elev= 30
    4347 1249.99  4383.5 1247.92  4389.7 1246.35  4418.9 1244.86  4438.9 1242.05
  4464.5 1240.78  4560.8 1235.45  4583.1 1232.84  4690.1 1226.52  4804.9 1223.57
  4919.7  1217.7  4940.5 1213.62  4946.7 1211.16  4955.1 1210.82  4982.2 1205.59
  4999.2 1204.43  4999.7 1203.93  5008.8 1204.43  5025.2 1205.73  5040.5 1205.42
  5054.7 1208.49  5113.6 1215.49  5150.2  1217.2  5192.6 1216.87  5265.7 1219.11
  5302.3 1221.67  5308.2 1221.08  5317.6 1222.73  5346.4 1224.62  5425.5 1226.51
#Mann= 8 ,-1 , 0
    4347     .12       0  4438.9     .05       0  4464.5     .12       0
  4583.1     .05       0  4999.2     .05       0  5008.8     .05       0
  5054.7     .12       0  5346.4     .05       0
Bank Sta=4999.2,5008.8
XS Rating Curve= 0 ,0
Exp/Cntr=0.3,0.1
