--- PECAN CREEK.prj (project) ---

Proj Title=PECAN CREEK Base Level Engineering
Current Plan=p01
Default Exp/Contr=0.3,0.1
English Units
Geom File=g01
Flow File=f01
Plan File=p01
Y Axis Title=Elevation
X Axis Title(PF)=Main Channel Distance
X Axis Title(XS)=Station
BEGIN DESCRIPTION:
PECAN CREEK
END DESCRIPTION:
DSS Export Rating Curves= 0
DSS Export Rating Curve Sorted= 0
DSS Export Volume Flow Curves= 0
DXF OffsetX= 0
DXF OffsetY= 0
DXF ScaleX= 1
DXF ScaleY= 10

--- PECAN CREEK.p01 (plan) ---

Plan Title=Multiple Run
Short Identifier=Multiple
Geom File=g01
Flow File=f01
Subcritical Flow
K Sum by GR= 0
Std Step Tol= 0.01
Critical Tol= 0.01
Num of Std Step Trials= 20
Max Error Tol= 0.3
Flow Tol Ratio= 0.001
Split Flow NTrial= 30
Split Flow Tol= 0.02
Split Flow Ratio= 0.02
Log Output Level= 0
Friction Slope Method= 1
Unsteady Friction Slope Method= 2
Unsteady Bridges Friction Slope Method= 1
Parabolic Critical Depth
Global Vel Dist=  1 , 1 , 1
Global Log Level= 0
CheckData=True
Encroach Param= -1, 0, 0, 0
BEGIN DESCRIPTION:
Multiple Run
END DESCRIPTION:

--- PECAN CREEK.f01 (steady flow) ---

Flow Title=Multiple
Program Version=4.10
Number of Profiles= 7
Profile Names=10-year,25-year,50-year,1pct_min,100-year,1pct_plu,500-year
River Rch & RM=PECAN CREEK,Reach-1         ,84013
    1300    2274    3065    2411    4235    7438    5791
River Rch & RM=PECAN CREEK,Reach-1         ,83500
    2468    4492    7174    5530   10230   18926   13929
River Rch & RM=PECAN CREEK,Reach-1         ,76500
    2973    5504    8923    6972   12824   23591   17461
River Rch & RM=PECAN CREEK,Reach-1         ,69500
    3100    5757    9410    7192   13551   25533   18459
River Rch & RM=PECAN CREEK,Reach-1         ,68000
    3637    6832   11232    8788   16250   30047   22114
River Rch & RM=PECAN CREEK,Reach-1         ,61000
    3780    7115   11696   10065   16929   28473   23013
River Rch & RM=PECAN CREEK,Reach-1         ,59500
    4011    7582   12423   10500   18010   30889   24479
River Rch & RM=PECAN CREEK,Reach-1         ,54661
    4874    9275   15181   11319   22013   42812   29713
River Rch & RM=PECAN CREEK,Reach-1         ,48500
    5202    9927   16177   14409   23474   38242   31645
River Rch & RM=PECAN CREEK,Reach-1         ,42000
    5462   10431   16975   18413   24625   32933   33137
River Rch & RM=PECAN CREEK,Reach-1         ,39930
   10312   19452   30847   26527   44074   73230   57779
River Rch & RM=PECAN CREEK,Reach-1         ,36944
   10462   19727   31188   23322   44547   85090   58355
River Rch & RM=PECAN CREEK,Reach-1         ,32000
   10779   20290   31860   27813   45430   74206   59367
River Rch & RM=PECAN CREEK,Reach-1         ,25000
   10713   20163   31603   30185   45053   67243   58851
River Rch & RM=PECAN CREEK,Reach-1         ,23646
   11211   21064   32920   26410   46865   83162   61116
River Rch & RM=PECAN CREEK,Reach-1         ,23168
   11779   22078   34296   26718   48724   88854   63374
River Rch & RM=PECAN CREEK,Reach-1         ,18000
   11897   22285   34566   26989   49081   89259   63798
River Rch & RM=PECAN CREEK,Reach-1         ,16500
   11865   22225   34454   27156   48921   88129   63585
River Rch & RM=PECAN CREEK,Reach-1         ,15000
   11884   22248   34421   27180   48855   87814   63461
River Rch & RM=PECAN CREEK,Reach-1         ,11052
   12112   22641   34906   27448   49479   89194   64176
River Rch & RM=PECAN CREEK,Reach-1         ,8546
   12306   22992   35428   27896   50201   90341   65087
River Rch & RM=PECAN CREEK,Reach-1         ,7854
   12109   22631   34861   27167   49409   89862   64071
River Rch & RM=PECAN CREEK,Reach-1         ,5926
   12364   23087   35512   27653   50300   91496   65179
River Rch & RM=PECAN CREEK,Reach-1         ,3417
   12730   23737   36431   28412   51542   93501   66705
Boundary for River Rch & Prof#=PECAN CREEK,Reach-1         , 1
Up Type= 0
Dn Type= 3
Dn Slope=0.001
Boundary for River Rch & Prof#=PECAN CREEK,Reach-1         , 2
Up Type= 0
Dn Type= 3
Dn Slope=0.001
Boundary for River Rch & Prof#=PECAN CREEK,Reach-1         , 3
Up Type= 0
Dn Type= 3
Dn Slope=0.001
Boundary for River Rch & Prof#=PECAN CREEK,Reach-1         , 4
Up Type= 0
Dn Type= 3
Dn Slope=0.001
Boundary for River Rch & Prof#=PECAN CREEK,Reach-1         , 5
Up Type= 0
Dn Type= 3
Dn Slope=0.001
Boundary for River Rch & Prof#=PECAN CREEK,Reach-1         , 6
Up Type= 0
Dn Type= 3
Dn Slope=0.001
Boundary for River Rch & Prof#=PECAN CREEK,Reach-1         , 7
Up Type= 0
Dn Type= 3
Dn Slope=0.001
DSS Import GetInterval= 0
DSS Import GetPeak= 0
DSS Import FillOption= 0

--- PECAN CREEK.g01 (geometry) ---

Geom Title=Existing Conditions
Program Version=4.10

River Reach=PECAN CREEK     ,Reach-1
Reach XY= 30
      2790221.75       10300209.      2790891.25       10297690.
      2793225.25       10297907.      2794810.25       10296043.
      2793527.25       10294742.        2795524.       10293823.
      2796361.25       10288608.       2797623.5       10287795.
        2797647.       10290283.      2799187.75       10288026.
        2797388.       10284691.      2798636.25       10284245.
      2799014.75       10281216.        2802842.       10277565.
        2802370.       10276332.       2803984.5       10275177.
      2804444.75       10272703.        2802206.       10271513.
       2802471.5       10268142.       2803478.5       10266605.
      2803311.25       10263309.       2804325.5       10261644.
        2804025.       10259703.        2806606.       10257459.
       2807007.5       10254364.      2809533.75       10252754.
      2809085.75       10250098.       2811754.5       10245214.
       2811456.5       10243510.      2812321.75       10242952.

Type RM Length L Ch R = 1 ,84013   ,513,513,513
BEGIN DESCRIPTION:
PECAN CREEK 168.0
END DESCRIPTION:
XS GIS Cut Line= 3
       2790727.8      10300296.8        2790240.       10300183.
       2789405.7     10299903.12
#Sta/Elev= 30
  4499.1 1442.18  4593.7 1433.24  4696.4 1428.69  4755.1 1423.86  4829.9 1421.09
  4881.2  1409.6    4893 1413.91  4930.5 1408.29  4978.1  1404.6  4983.9 1402.22
  5009.8 1400.69  5010.3 1400.19  5025.9 1400.69  5036.2 1401.62  5044.1  1404.9
  5049.4 1403.84  5122.9 1409.72  5170.3 1414.07  5214.4  1416.1  5327.9 1416.75
  5415.9 1418.25  5533.3 1417.61  5554.1 1417.07  5643.4 1422.06    5675 1422.42
  5711.8 1428.92  5738.1 1436.23  5765.7 1440.91  5813.7 1452.07    5880  1466.1
#Mann= 9 ,-1 , 0
  4499.1     .05       0  5009.8     .05       0  5025.9     .05       0
  5122.9     .12       0  5214.4     .05       0  5327.9     .12       0
  5533.3     .05       0  5765.7     .12       0  5813.7     .05       0
Bank Sta=5009.8,5025.9
XS Rating Curve= 0 ,0
Exp/Cntr=0.3,0.1

Type RM Length L Ch R = 1 ,83500   ,500,500,500
BEGIN DESCRIPTION:
PECAN CREEK 167.0
END DESCRIPTION:
XS GIS Cut Line= 3
      2790505.67      10300003.1       2790125.5     10299736.21
      2789605.68     10299853.11
#Sta/Elev= 30
  4535.5 1432.14  4575.4 1427.24  4694.3 1417.79  4730.2 1411.98  4736.4  1409.5
  4751.2 1407.92  4801.7 1404.86  4842.7 1404.21  4858.4 1404.86  4908.9 1402.39
  4959.4 1402.69  4980.9 1400.18  4987.9  1396.9  4988.4  1396.4  5008.7  1396.9
  5020.3 1399.94  5060.9 1403.86  5085.6 1409.46  5098.5 1412.98  5103.6 1410.89
  5112.6 1412.81  5174.1 1414.68  5290.1 1413.66  5392.4 1415.05  5436.6 1416.24
  5465.3 1418.24  5471.3 1419.68  5508.6 1423.24  5513.7 1422.69  5532.8 1425.26
#Mann= 11 ,-1 , 0
  4535.5     .05       0  4575.4     .12       0  4842.7     .05       0
  4980.9     .12       0  4987.9     .07       0  5008.7     .12       0
  5060.9     .05       0  5085.6     .12       0  5290.1     .05       0
  5392.4     .12       0  5436.6     .05       0
Bank Sta=4987.9,5008.7
XS Rating Curve= 0 ,0
Exp/Cntr=0.3,0.1

Type RM Length L Ch R = 1 ,83000   ,500,500,500
BEGIN DESCRIPTION:
PECAN CREEK 166.0
END DESCRIPTION:
XS GIS Cut Line= 3
      2790755.66     10299403.11       2790333.5     10299291.38
      2790155.66     10299103.08
#Sta/Elev= 30
  4563.3 1432.07  4580.8 1429.84    4586 1430.31  4604.7 1428.34  4661.3 1425.17
  4741.7 1418.14  4832.2 1406.64  4925.3 1401.65    4946 1397.47  4974.5 1397.89
    4978 1397.93  4985.8 1394.26  4986.3 1393.76  5006.8 1394.26  5025.3 1398.36
  5046.8 1400.74  5053.7 1403.78  5075.1  1404.9    5082 1404.23  5089.3 1401.71
  5117.6    1406  5125.8 1408.77  5138.6 1411.06  5145.9 1410.06  5152.8 1411.09
  5174.2 1411.13  5181.1 1412.38  5188.4 1412.02  5223.6 1414.54    5259 1418.17
#Mann= 5 ,-1 , 0
  4563.3     .12       0  4974.5     .05       0  4985.8     .05       0
  5006.8     .05       0  5125.8     .12       0
Bank Sta=4985.8,5006.8
XS Rating Curve= 0 ,0
Exp/Cntr=0.3,0.1

Type RM Length L Ch R = 1 ,82500   ,500,500,500
BEGIN DESCRIPTION:
PECAN CREEK 165.0
END DESCRIPTION:
XS GIS Cut Line= 3
      2790705.68     10298753.11      2790476.47     10298824.59
      2790255.71      10298903.1
#Sta/Elev= 30
  4759.9 1418.37  4791.3 1414.46  4808.7  1410.4  4813.9 1410.58  4841.2 1402.55
  4846.4 1403.02  4863.5  1401.1  4885.6 1399.95    4938 1399.55  4943.9 1397.92
  4949.2 1398.11  4958.9 1396.56  4969.4 1394.05  4976.4 1391.11  4981.7 1392.42
  4987.3 1391.05  4987.8 1390.55  5008.3 1391.05  5039.2 1395.56  5044.5 1395.38
    5070 1401.35  5075.3 1400.77  5105.4  1405.4  5157.2 1409.78  5162.5  1409.4
  5188.1 1413.59  5193.4  1413.1  5211.9 1415.64  5218.9 1416.78  5234.3 1416.81
#Mann= 6 ,-1 , 0
  4759.9     .05       0  4863.5     .12       0  4987.3     .05       0
  5008.3     .12       0  5105.4     .12       0  5211.9     .05       0
Bank Sta=4987.3,5008.3
XS Rating Curve= 0 ,0
Exp/Cntr=0.3,0.1

Type RM Length L Ch R = 1 ,82000   ,500,500,500
BEGIN DESCRIPTION:
PECAN CREEK 164.0
END DESCRIPTION:
XS GIS Cut Line= 3
       2790905.7     10298603.13      2790646.86     10298360.77
      2790155.65      10298153.1
#Sta/Elev= 30
  4645.4 1417.83  4666.7 1417.33  4701.9 1414.96  4709.2 1415.69    4716 1414.06
  4765.8 1412.36  4871.8 1404.32  4900.2  1398.6  4921.2 1398.03  4935.3 1395.98
  4942.7 1393.81  4977.8 1389.65  4981.5 1387.08    4982 1386.58  5002.6 1387.08
  5003.4 1388.45  5012.2 1389.35  5030.5 1394.96  5044.7 1396.71  5119.4 1400.73
  5165.2 1402.46  5312.8 1413.18  5336.5 1414.05  5381.3 1419.67    5403 1423.44
  5435.6    1427  5465.9 1431.85  5489.6 1433.58  5533.1 1438.38  5533.3 1438.38
#Mann= 5 ,-1 , 0
  4645.4     .12       0  4981.5     .07       0  5002.6     .12       0
  5119.4     .05       0  5533.1     .12       0
Bank Sta=4981.5,5002.6
XS Rating Curve= 0 ,0
Exp/Cntr=0.3,0.1

Type RM Length L Ch R = 1 ,81500   ,500,500,500
BEGIN DESCRIPTION:
PECAN CREEK 163.0
END DESCRIPTION:
XS GIS Cut Line= 3
      2791205.71     10298303.14      2790790.59     10297886.85
       2790455.7     10298003.11
#Sta/Elev= 30
  4412.1 1415.64  4426.3 1415.52  4447.5 1412.94  4565.3 1407.62  4702.1 1403.11
  4709.1 1401.76  4750.8 1401.34  4850.5 1397.89  4878.8 1395.49  4942.5 1392.88
  4949.5 1391.09  4970.8 1389.01  4988.3 1385.85  4988.8 1385.35  5009.7 1385.85
  5015.8 1388.36  5029.6  1390.6  5064.1 1394.67  5157.5 1398.89  5183.3 1404.39
  5186.6 1404.23  5238.1 1409.72  5245.6 1411.66  5250.9 1410.78  5269.8 1414.63
  5276.7 1417.04    5282 1416.68    5291 1419.59  5341.6  1424.4  5354.5 1425.22
#Mann= 8 ,-1 , 0
  4412.1     .12       0  4565.3     .05       0  4750.8     .12       0
  4988.3     .07       0  5009.7     .12       0  5029.6     .05       0
  5186.6     .12       0  5341.6     .05       0
Bank Sta=4988.3,5009.7
XS Rating Curve= 0 ,0
Exp/Cntr=0.3,0.1

Type RM Length L Ch R = 1 ,81000   ,500,500,500
BEGIN DESCRIPTION:
PECAN CREEK 162.0
END DESCRIPTION:
XS GIS Cut Line= 3
      2791505.68     10298403.09      2791140.85     10297606.24
      2791105.69     10297403.16
#Sta/Elev= 30
  4123.6 1444.24  4258.4 1426.05  4298.9 1423.45  4304.4 1421.68  4355.9 1416.94
  4401.9 1410.37  4437.9 1408.14  4486.5 1402.43  4509.7 1401.15  4568.5 1400.09
  4637.2 1396.78  4747.4 1393.33  4884.1  1390.3  4893.5 1389.77  4901.6 1387.67
  4937.4 1386.25  4981.7 1386.72  4988.2 1383.73  4988.7 1383.23  5009.7 1383.73
  5033.6 1385.39  5053.9 1390.55  5059.3 1397.31  5064.4 1397.88  5074.2 1403.18
  5084.4  1406.6  5119.1  1412.1  5155.4 1421.48  5171.5 1422.72  5206.1 1425.04
#Mann= 8 ,-1 , 0
  4123.6     .12       0  4437.9     .05       0  4509.7     .12       0
  4637.2     .05       0  4747.4     .12       0  4988.2     .07       0
  5009.7     .12       0  5171.5     .05       0
Bank Sta=4988.2,5009.7
XS Rating Curve= 0 ,0
Exp/Cntr=0.3,0.1

Type RM Length L Ch R = 1 ,80500   ,500,500,500
BEGIN DESCRIPTION:
PECAN CREEK 161.0
END DESCRIPTION:
XS GIS Cut Line= 3
      2791655.69     10298103.14      2791555.94     10297861.41
      2791355.69     10297353.14
#Sta/Elev= 30
  4738.5  1418.9    4771 1414.95  4830.4 1403.59  4878.2  1398.6  4931.5  1390.5
  4960.8 1382.54  4966.2 1383.03  4982.2 1380.58  5008.9 1379.82  5009.4 1379.32
  5030.4 1379.82  5044.1 1380.36  5068.5 1383.99  5098.2 1385.27  5119.8 1384.92
  5137.9 1385.07  5170.1  1388.1  5176.8 1390.22  5182.1 1390.02  5201.2  1393.8
  5206.5 1393.54  5213.1 1395.49  5228.1 1396.95  5290.5 1399.69  5393.4 1407.81
  5447.5 1409.43  5452.9 1411.12  5471.1 1411.62  5502.1 1415.06  5546.3 1419.18
#Mann= 7 ,-1 , 0
  4738.5     .12       0  4982.2     .05       0  5008.9     .05       0
  5030.4     .05       0  5119.8     .12       0  5228.1     .05       0
  5502.1     .12       0
Bank Sta=5008.9,5030.4
XS Rating Curve= 0 ,0
Exp/Cntr=0.3,0.1

Type RM Length L Ch R = 1 ,80000   ,500,500,500
BEGIN DESCRIPTION:
PECAN CREEK 160.0
END DESCRIPTION:
XS GIS Cut Line= 3
      2792105.68     10297903.11      2792022.83       10297795.
      2792255.67     10297303.13
#Sta/Elev= 30
  4863.8 1400.52  4885.6 1395.55  4914.2 1392.21  4939.7 1386.77  4949.9  1384.5
  4956.2  1385.1  4964.5 1380.06  4977.2  1377.7  4980.8  1374.4  4981.3  1373.9
  5002.4  1374.4  5003.8 1375.36  5018.5 1374.49    5064 1378.74  5107.6 1380.15
  5123.8 1380.31    5155  1383.5  5160.6 1382.33  5183.3 1383.69  5200.5 1386.64
  5245.5 1388.96  5267.6 1392.09  5400.4 1419.99  5414.4 1421.65  5439.1 1424.68
  5445.1 1424.09  5484.6 1424.46  5490.1 1425.99  5507.3 1426.22  5544.2 1430.92
#Mann= 7 ,-1 , 0
  4863.8     .12       0  4939.7     .05       0  4980.8     .07       0
  5002.4     .05       0  5107.6     .05       0  5414.4     .12       0
  5445.1     .05       0
Bank Sta=4980.8,5002.4
XS Rating Curve= 0 ,0
Exp/Cntr=0.3,0.1

Type RM Length L Ch R = 1 ,79500   ,500,500,500
BEGIN DESCRIPTION:
PECAN CREEK 159.0
END DESCRIPTION:
XS GIS Cut Line= 3
      2792305.66     10298053.15      2792500.56       10297657.
      2792605.69     10297453.11
#Sta/Elev= 30
  4558.5 1410.46  4638.6 1401.21  4662.5 1397.53  4707.4 1394.07  4742.7 1389.89
  4836.7 1382.99  4864.7 1381.99  4870.6 1380.44  4926.3 1376.39  4932.1    1375
  4946.5 1375.01  4954.6 1373.24  4982.6 1371.67  4988.6 1369.84  4989.1 1369.34
  5010.2 1369.84  5027.3 1373.88  5038.1 1377.61  5043.8 1385.59  5049.5 1386.09
  5060.4 1392.75    5066 1393.34  5071.9  1401.1  5088.2 1405.84  5139.4 1414.48
  5171.2  1418.2  5176.8  1419.8  5193.3 1419.95  5206.8 1421.49  5229.4  1422.8
#Mann= 7 ,-1 , 0
  4558.5     .05       0  4638.6     .12       0  4742.7     .05       0
  4946.5     .12       0  4988.6     .07       0  5010.2     .12       0
  5206.8     .05       0
Bank Sta=4988.6,5010.2
XS Rating Curve= 0 ,0
Exp/Cntr=0.3,0.1

Type RM Length L Ch R = 1 ,79000   ,500,500,500
BEGIN DESCRIPTION:
PECAN CREEK 158.0
END DESCRIPTION:
XS GIS Cut Line= 3
       2793355.7     10298203.13      2792967.59     10297812.86
      2792905.69     10297453.15
#Sta/Elev= 30
  4449.6 1444.48  4555.7 1433.61    4591 1426.97  4598.1 1423.67  4605.2 1423.23
  4626.4 1412.22  4633.5 1411.04  4640.5 1406.33  4661.7 1401.79    4683 1393.28
    4690 1392.74  4697.1 1388.76  4725.4 1380.99  4749.5 1378.43  4824.4 1371.79
  4845.6 1372.17  4852.7 1369.73  4859.7 1370.98  4866.8 1368.43  4873.9 1369.56
  4902.2 1366.53  4916.3 1368.21    4969 1366.35  4969.5 1365.85  4990.9 1366.35
  5043.1 1371.08  5101.5 1382.64  5201.9 1395.57  5354.4 1422.65    5365 1423.67
#Mann= 7 ,-1 , 0
  4449.6     .12       0  4749.5     .05       0    4969     .03       0
  4990.9     .05       0  5101.5     .12       0  5201.9     .05       0
  5354.4     .12       0
Bank Sta=4969,4990.9
XS Rating Curve= 0 ,0
Exp/Cntr=0.3,0.1

Type RM Length L Ch R = 1 ,78500   ,500,500,500
BEGIN DESCRIPTION:
PECAN CREEK 157.0
END DESCRIPTION:
XS GIS Cut Line= 3
      2793505.67      10297853.1      2793380.85     10297758.52
      2792905.67      10297403.1
#Sta/Elev= 30
  4843.4 1419.11  4846.5 1419.11  4865.2 1413.97  4871.5  1411.3  4879.8 1409.69
  4902.9 1401.11  4906.9 1398.79  4915.1 1396.87    4936 1389.16  4956.8 1375.99
  4979.6 1365.72  4982.9 1363.11  4983.4 1362.61  5004.8 1363.11    5015 1365.34
  5065.1 1370.16  5079.6 1371.17  5085.9 1370.49    5105 1373.96  5166.9 1379.84
  5229.7 1384.46  5243.7  1384.5    5386 1397.35  5429.8    1403    5486 1408.65
  5523.2 1414.92  5565.2 1421.98  5571.5 1420.77  5582.7 1421.21  5593.4 1421.44
#Mann= 8 ,-1 , 0
  4843.4     .12       0  4902.9     .05       0  4982.9     .05       0
  5004.8     .05       0    5105     .12       0  5166.9     .05       0
  5523.2     .12       0  5582.7     .05       0
Bank Sta=4982.9,5004.8
XS Rating Curve= 0 ,0
Exp/Cntr=0.3,0.1

Type RM Length L Ch R = 1 ,78000   ,500,500,500
BEGIN DESCRIPTION:
PECAN CREEK 156.0
END DESCRIPTION:
XS GIS Cut Line= 3
      2793805.68      10297553.1      2793562.18     10297302.38
      2793055.69     10296803.11
#Sta/Elev= 30
  4650.5 1418.53  4678.7 1414.13    4700 1409.72  4721.1 1403.33  4793.3 1389.52
  4804.1  1386.9  4841.5 1379.41  4862.6 1372.08  4876.7 1368.67  4890.6 1367.31
  4933.3 1361.94  4982.9 1362.91  4993.1 1360.66  4993.6 1360.16    5015 1360.66
  5018.2 1364.63  5039.4 1368.42    5074 1370.12  5080.9 1370.71  5173.8 1378.59
  5357.7  1386.9  5421.4 1394.35  5442.5 1396.41  5503.9 1405.94  5534.4 1412.47
  5559.8 1414.61    5584  1416.5  5619.3 1422.21    5683 1429.67  5711.2 1435.08
#Mann= 11 ,-1 , 0
  4650.5     .05       0  4793.3     .12       0  4804.1     .05       0
  4890.6     .12       0  4993.1     .07       0    5015     .12       0
    5074     .05       0  5080.9     .12       0  5421.4     .05       0
  5503.9     .12       0  5559.8     .05       0
Bank Sta=4993.1,5015
XS Rating Curve= 0 ,0
Exp/Cntr=0.3,0.1

Type RM Length L Ch R = 1 ,77500   ,500,500,500
BEGIN DESCRIPTION:
PECAN CREEK 155.0
END DESCRIPTION:
XS GIS Cut Line= 3
       2794055.7     10297103.13       2793813.7     10296873.23
      2793305.72     10296503.14
#Sta/Elev= 30
  4666.2 1406.59  4708.5 1400.96  4722.7 1397.01  4768.4 1388.53  4800.7 1383.05
  4843.2 1373.32  4864.2 1370.67  4892.5 1364.18    4935 1361.35  4949.2 1357.45
  4970.2 1359.73  4984.4 1358.33  4985.5 1356.29    4986 1355.79  5007.4 1356.29
  5034.7 1363.19  5056.4 1365.56  5077.3 1364.83    5092 1367.45  5163.1 1371.44
    5299 1381.85  5343.1 1389.02  5370.1 1395.43  5393.3 1399.01  5420.3 1405.85
  5449.7 1410.35  5492.4 1422.71  5529.3 1426.86    5571  1435.1  5628.5 1442.54
#Mann= 4 ,-1 , 0
  4666.2     .12       0  4768.4     .05       0  4985.5     .05       0
  5007.4     .05       0
Bank Sta=4985.5,5007.4
XS Rating Curve= 0 ,0
Exp/Cntr=0.3,0.1

Type RM Length L Ch R = 1 ,77000   ,500,500,500
BEGIN DESCRIPTION:
PECAN CREEK 154.0
END DESCRIPTION:
XS GIS Cut Line= 3
      2794155.69     10296853.15      2794052.27     10296435.67
      2794005.69     10296253.12
#Sta/Elev= 30
  4569.9 1388.59  4611.1 1384.18  4643.5 1379.68  4683.3 1374.71  4698.3 1373.73
  4712.3 1371.99  4753.6 1369.37  4765.7  1367.8  4848.1 1362.11  4868.7 1361.32
  4909.9 1354.17  4930.5 1355.04  4960.6 1354.67  5022.6 1352.71  5023.1 1352.21
  5044.1 1352.21  5044.6 1352.71    5048 1356.19  5054.2 1355.94  5083.7 1359.81
  5088.8 1361.55  5105.8 1364.78  5124.5  1370.4  5129.7 1370.33  5136.8 1372.98
  5162.6  1378.5  5165.4 1379.62  5170.6 1379.59  5185.8 1384.61  5188.4 1384.61
#Mann= 6 ,-1 , 0
  4569.9     .12       0  4643.5     .05       0  4698.3     .12       0
  4848.1     .05       0  5022.6     .05       0  5044.6     .05       0
Bank Sta=5022.6,5044.6
XS Rating Curve= 0 ,0
Exp/Cntr=0.3,0.1

Type RM Length L Ch R = 1 ,76500   ,500,500,500
BEGIN DESCRIPTION:
PECAN CREEK 153.0
END DESCRIPTION:
XS GIS Cut Line= 3
      2794905.68     10296653.11        2794488.      10296236.4
      2794455.69     10296053.12
#Sta/Elev= 30
    4410 1385.73  4461.5 1381.43  4642.6 1367.42  4664.5 1366.53  4685.8 1363.62
  4721.1 1364.24  4777.7 1360.96  4798.9 1357.19    4806 1357.48    4813 1354.92
  4820.1 1356.13  4827.2 1351.93  4834.2 1352.98  4876.7 1350.99  4883.8 1351.99
  4890.8 1350.61  4897.9 1354.13    4905 1352.46    4912 1355.62  4926.2 1355.73
  4950.8 1352.86  4975.7 1350.83  4978.2 1348.84  4978.7 1348.34  5001.5 1348.84
  5033.8 1352.67  5054.1 1362.06  5084.6  1370.2  5145.5 1378.91  5186.1 1380.38
#Mann= 6 ,-1 , 0
    4410     .12       0  4461.5     .05       0  4642.6     .12       0
  4950.8     .05       0  4978.2     .05       0  5001.5     .05       0
Bank Sta=4978.2,5001.5
XS Rating Curve= 0 ,0
Exp/Cntr=0.3,0.1

Type RM Length L Ch R = 1 ,76000   ,500,500,500
BEGIN DESCRIPTION:
PECAN CREEK 152.0
END DESCRIPTION:
XS GIS Cut Line= 3
      2795105.72     10295903.11      2794853.93     10295937.27
       2794505.7     10295903.11
#Sta/Elev= 30
  4745.9 1410.52  4748.6 1410.49  4776.2 1402.91  4782.2 1399.51  4787.2 1400.57
  4854.7 1364.13  4859.7 1364.83    4867    1362  4877.1  1360.3  4917.5 1356.53
  4927.2 1354.95  4947.8 1354.66  4957.9 1353.67    4978 1350.02    5000 1348.68
  5006.6 1347.56  5007.1 1347.06    5030 1347.56  5038.4 1350.66  5048.5 1351.26
  5068.6  1350.5  5098.8 1351.03  5130.3 1354.31  5157.5 1357.42    5169 1359.81
  5219.3  1364.6  5296.7 1369.81  5301.7    1369  5319.8 1370.71  5349.9 1371.89
#Mann= 6 ,-1 , 0
  4745.9     .12       0  4748.6     .05       0  5006.6     .05       0
    5030     .05       0  5130.3     .12       0  5157.5     .05       0
Bank Sta=5006.6,5030
XS Rating Curve= 0 ,0
Exp/Cntr=0.3,0.1

Type RM Length L Ch R = 1 ,75500   ,500,500,500
BEGIN DESCRIPTION:
PECAN CREEK 151.0
END DESCRIPTION:
XS GIS Cut Line= 3
      2794805.69      10295353.1      2794699.89     10295530.91
      2794355.71     10295953.08
#Sta/Elev= 30
  4793.1 1413.59  4816.4 1409.06  4843.7 1399.83  4874.6 1385.36  4880.7 1379.64
  4886.6 1376.02  4902.2 1361.21  4909.5 1348.66  4923.6 1342.96  4932.7 1342.81
  4939.2 1344.21    4945 1344.14  4960.6 1342.92    4982 1342.85  4985.9 1341.87
  4986.4 1341.37  5009.3 1341.87  5026.3 1345.09  5040.7 1345.99  5054.5  1349.4
  5067.9  1350.8  5090.2 1352.41  5182.8 1354.48  5196.4 1356.23  5238.8 1358.52
  5302.7 1364.11  5331.5  1365.6  5352.3 1368.06  5424.1 1373.76  5544.7 1382.27
#Mann= 3 ,-1 , 0
  4793.1     .12       0  4985.9     .05       0  5009.3     .05       0
Bank Sta=4985.9,5009.3
XS Rating Curve= 0 ,0
Exp/Cntr=0.3,0.1

Type RM Length L Ch R = 1 ,75000   ,500,500,500
BEGIN DESCRIPTION:
PECAN CREEK 150.0
END DESCRIPTION:
XS GIS Cut Line= 3
      2794605.69     10295153.11       2794229.4      10295375.9
      2793705.67     10295603.12
#Sta/Elev= 30
  4562.7 1401.16  4583.5 1398.52  4650.5 1389.32  4703.9 1383.88    4737 1378.46
  4767.4 1370.82  4783.1 1368.49  4876.5 1346.31  4911.7 1343.87  4964.4 1343.62
    4980 1342.15  4987.6 1339.41  4988.1 1338.91    5011 1339.41    5015 1341.29
  5091.3  1340.7  5106.8 1344.39  5135.7 1347.75  5222.1 1354.24  5253.1 1359.93
    5282 1362.94  5310.9 1368.53  5374.7 1376.72  5428.2 1386.53  5433.7 1389.18
  5457.1 1394.06    5486 1398.91  5509.5 1401.03    5533 1406.15  5570.9 1411.87
#Mann= 5 ,-1 , 0
  4562.7     .05       0  4583.5     .12       0  4703.9     .05       0
  4987.6     .05       0    5011     .05       0
Bank Sta=4987.6,5011
XS Rating Curve= 0 ,0
Exp/Cntr=0.3,0.1

Type RM Length L Ch R = 1 ,74500   ,500,500,500
BEGIN DESCRIPTION:
PECAN CREEK 149.0
END DESCRIPTION:
XS GIS Cut Line= 3
       2794055.7     10294903.09      2793813.46     10295127.19
       2793605.7     10295503.09
#Sta/Elev= 30
    4670 1361.29  4712.3 1359.08    4833 1343.96  4880.2 1340.34  4958.9  1336.2
  4967.4 1337.39  4991.6 1334.51  4992.1 1334.01  5015.1 1334.51  5025.2 1338.69
  5046.9 1342.98  5068.7 1343.79    5150 1352.63  5166.1 1356.69  5187.8 1365.98
  5193.5 1369.94  5209.6 1373.28  5215.3 1377.24  5231.4 1380.72  5237.1 1384.94
  5253.1 1387.84  5258.8 1391.14  5290.9 1395.73  5296.2 1398.36  5312.7 1399.35
  5318.4 1401.51  5334.5    1403    5378 1411.58  5405.9 1415.09  5429.5  1419.6
#Mann= 7 ,-1 , 0
    4670     .05       0  4880.2     .12       0  4958.9     .05       0
  4991.6     .03       0  5015.1     .05       0  5296.2     .12       0
  5405.9     .05       0
Bank Sta=4991.6,5015.1
XS Rating Curve= 0 ,0
Exp/Cntr=0.3,0.1

Type RM Length L Ch R = 1 ,74000   ,500,500,500
BEGIN DESCRIPTION:
PECAN CREEK 148.0
END DESCRIPTION:
XS GIS Cut Line= 3
      2794305.66      10294953.1      2793529.94     10294732.79
      2793455.69     10294553.13
#Sta/Elev= 30
  4193.6 1375.92  4283.5 1370.88  4370.3 1362.75  4429.5 1362.75  4513.6 1353.76
  4614.5 1344.84  4642.4 1344.31  4786.1  1337.2  4817.3 1338.64  4856.7 1335.01
  4859.6 1334.92  4879.7  1332.1  4973.2 1332.98  4982.2 1329.48  4982.7 1328.98
  5005.9 1329.48  5020.1  1331.3  5032.1 1338.68  5051.7 1356.78  5054.8 1360.84
  5086.2 1380.98  5102.6 1384.82    5108 1388.38  5126.5 1389.33  5131.9 1391.68
  5152.2 1394.49  5155.8 1396.38  5179.8 1395.29  5185.2 1397.75  5194.4 1398.09
#Mann= 9 ,-1 , 0
  4193.6     .05       0  4513.6     .12       0  4642.4     .05       0
  4856.7     .12       0  4859.6     .05       0  4982.2     .05       0
  5005.9     .05       0  5051.7     .12       0  5152.2     .05       0
Bank Sta=4982.2,5005.9
XS Rating Curve= 0 ,0
Exp/Cntr=0.3,0.1

Type RM Length L Ch R = 1 ,73500   ,500,500,500
BEGIN DESCRIPTION:
PECAN CREEK 147.0
END DESCRIPTION:
XS GIS Cut Line= 3
      2794055.67     10294853.07      2793977.39     10294588.92
      2793905.67     10294403.08
#Sta/Elev= 30
  4724.5 1359.53  4733.6 1359.01  4807.6 1350.38  4812.8 1349.53  4818.3 1346.85
  4839.2 1345.55  4851.2 1343.45  4870.5 1341.63  4879.3 1339.18  4912.2 1334.64
  4917.7 1332.42  4983.3 1326.34  4983.8 1325.84  5007.1 1326.34  5015.1  1328.2
  5027.7 1328.73  5038.4  1330.3  5045.1 1332.48  5059.8 1334.68  5069.7 1340.66
  5074.5 1345.67  5081.3 1350.24    5092 1353.62  5099.6 1359.85  5113.4 1367.62
  5124.1 1371.36    5135 1377.44    5167 1388.91  5189.5 1395.06  5199.2 1396.15
#Mann= 5 ,-1 , 0
  4724.5     .05       0  4733.6     .12       0  4983.3     .05       0
  5007.1     .12       0  5074.5     .12       0
Bank Sta=4983.3,5007.1
XS Rating Curve= 0 ,0
Exp/Cntr=0.3,0.1

Type RM Length L Ch R = 1 ,73000   ,500,500,500
BEGIN DESCRIPTION:
PECAN CREEK 146.0
END DESCRIPTION:
XS GIS Cut Line= 3
      2794405.68     10294903.14      2794454.71     10294481.88
       2794255.7     10294153.13
#Sta/Elev= 30
  4575.9 1372.13  4615.2 1367.63  4620.2 1368.79  4626.3 1366.51  4650.4 1363.33
  4703.7  1354.9  4708.8 1356.46  4777.3 1345.16  4787.2 1344.16  4797.4 1345.59
  4847.8 1339.09  4908.2 1336.06  4945.6  1331.7  4958.5 1330.74  4964.3 1327.83
  4969.4 1329.76    4985 1321.99  4985.5 1321.49  5008.8 1321.99  5033.6 1327.69
  5048.8  1329.5  5070.1 1328.06  5092.1 1324.36  5122.5 1331.65  5170.6 1337.58
  5240.9 1358.74  5288.5 1373.12  5325.9 1384.15  5339.7 1390.41  5384.3 1400.06
#Mann= 8 ,-1 , 0
  4575.9     .12       0  4650.4     .05       0  4945.6     .12       0
    4985     .07       0  5008.8     .12       0  5170.6     .05       0
  5240.9     .12       0  5288.5     .05       0
Bank Sta=4985,5008.8
XS Rating Curve= 0 ,0
Exp/Cntr=0.3,0.1

Type RM Length L Ch R = 1 ,72500   ,500,500,500
BEGIN DESCRIPTION:
PECAN CREEK 145.0
END DESCRIPTION:
XS GIS Cut Line= 3
      2795155.68     10294503.11      2794892.08     10294255.58
      2794705.69     10294053.11
#Sta/Elev= 30
  4638.4 1358.67  4723.1 1351.93  4815.4 1340.44  4850.6 1334.09  4921.4 1326.04
  4935.6 1326.86  4942.5 1325.93  4949.8 1326.94  4956.6 1325.25  4963.9 1326.76
  4970.8 1325.44  4978.2  1325.6  4992.2  1320.7  5020.3 1321.86  5022.6 1320.37
  5023.1 1319.87  5046.4 1320.37  5062.8 1324.08  5091.2 1326.74  5112.2 1330.78
  5119.5 1334.71  5126.3 1335.93  5147.9 1343.18    5183  1351.5  5204.6 1358.83
  5234.2 1366.62  5261.3 1371.24  5268.1 1370.75  5271.3 1371.86  5275.2 1372.03
#Mann= 6 ,-1 , 0
  4638.4     .05       0  4978.2     .12       0  5022.6     .07       0
  5046.4     .12       0  5234.2     .05       0  5271.3     .12       0
Bank Sta=5022.6,5046.4
XS Rating Curve= 0 ,0
Exp/Cntr=0.3,0.1

Type RM Length L Ch R = 1 ,72000   ,500,500,500
BEGIN DESCRIPTION:
PECAN CREEK 144.0
END DESCRIPTION:
XS GIS Cut Line= 3
       2795455.7     10294153.13      2795342.91     10294047.83
      2794855.68     10293853.11
#Sta/Elev= 30
  4845.7 1348.12  4849.1 1348.12  4859.6 1345.41  4881.1  1343.3    4931 1334.79
    4952 1330.91  4966.1  1326.9    4973  1323.7  4987.2 1319.62  4987.8 1317.26
  4988.3 1316.76  5011.7 1317.26  5018.6 1319.32  5025.1 1320.03  5054.7 1319.26
  5084.3 1324.41  5103.2 1324.24  5180.1 1328.13  5225.2  1331.8  5240.5 1332.59
  5264.8 1335.49  5299.8 1343.37  5318.7 1346.21  5353.7 1354.12  5363.2 1355.41
  5407.5 1366.17    5456 1375.03  5509.9 1382.73  5515.3 1381.47  5524.7 1382.27
#Mann= 5 ,-1 , 0
  4845.7     .05       0    4931     .12       0  4987.8     .07       0
  5011.7     .12       0  5225.2     .05       0
Bank Sta=4987.8,5011.7
XS Rating Curve= 0 ,0
Exp/Cntr=0.3,0.1

Type RM Length L Ch R = 1 ,71500   ,500,500,500
BEGIN DESCRIPTION:
PECAN CREEK 143.0
END DESCRIPTION:
XS GIS Cut Line= 3
      2795955.67     10293703.11      2795578.35     10293624.13
       2795355.7     10293553.12
#Sta/Elev= 30
  4614.5 1395.88  4634.4 1392.69  4639.5 1392.94  4675.8 1386.63  4684.3 1384.26
  4689.4 1384.22    4778  1361.7  4784.2 1359.37  4816.4  1352.4  4834.1 1348.49
  4839.3 1345.44  4869.9 1337.64    4879  1334.4  4884.1 1334.64  4900.6 1326.68
  4912.7 1323.01  4928.9 1319.43  4941.4 1318.01  4972.1 1317.45  4978.9 1316.78
  4980.5 1315.63    4981 1315.13  5004.5 1315.63  5051.4 1320.82  5139.3 1324.29
  5170.7 1332.21  5180.2 1333.85  5185.4 1332.41  5202.2 1334.34  5233.7 1340.63
#Mann= 5 ,-1 , 0
  4614.5     .05       0  4816.4     .12       0  4912.7     .05       0
  4980.5     .05       0  5004.5     .05       0
Bank Sta=4980.5,5004.5
XS Rating Curve= 0 ,0
Exp/Cntr=0.3,0.1

Type RM Length L Ch R = 1 ,71000   ,500,500,500
BEGIN DESCRIPTION:
PECAN CREEK 142.0
END DESCRIPTION:
XS GIS Cut Line= 3
      2795755.68     10293253.11      2795525.34     10293137.99
      2795005.71     10292653.14
#Sta/Elev= 30
  4742.5 1361.82  4783.1 1355.42  4845.9 1343.34  4890.6 1329.56  4907.4 1322.35
    4913 1323.68  4929.8 1317.48  4935.4 1319.12  4952.1 1313.66  4957.7 1315.37
  4966.1 1311.37  4984.8 1308.12  4985.3 1307.62  5008.9 1308.12  5044.7  1308.8
  5109.1 1310.77  5144.8 1314.31  5208.3 1315.42  5231.8 1318.31  5264.9 1321.81
  5328.5 1335.66  5385.1 1343.64    5435 1355.93  5486.5 1363.27  5519.5 1370.22
  5547.8 1370.89  5597.6 1379.22  5648.5 1385.19  5682.6 1391.26  5710.7 1399.18
#Mann= 8 ,-1 , 0
  4742.5     .12       0  4783.1     .05       0  4984.8     .05       0
  5008.9     .05       0  5044.7     .12       0  5231.8     .05       0
  5486.5     .12       0  5648.5     .05       0
Bank Sta=4984.8,5008.9
XS Rating Curve= 0 ,0
Exp/Cntr=0.3,0.1

Type RM Length L Ch R = 1 ,70500   ,500,500,500
BEGIN DESCRIPTION:
PECAN CREEK 141.0
END DESCRIPTION:
XS GIS Cut Line= 3
      2795955.67      10293153.1       2795556.1     10292776.18
       2795355.7     10292703.12
#Sta/Elev= 30
  4450.7 1369.08  4486.1 1363.94    4493    1365  4500.2  1362.6  4507.1 1363.98
  4514.4 1361.43  4549.6 1359.19  4620.4 1342.15  4684.3 1334.59  4691.2 1331.93
  4733.7 1328.21  4740.6 1325.47  4889.4  1315.2  4924.6 1310.55  4938.8 1311.44
  4945.7 1308.52    4953 1310.28  4959.8 1306.29  4967.1 1309.07    4974 1305.55
  4986.5 1305.39    4987 1304.89  5010.6 1305.39  5081.1 1307.57  5106.3 1323.94
  5111.7 1322.93  5117.5  1329.7  5149.5 1342.11  5181.4 1346.53  5213.3 1345.32
#Mann= 3 ,-1 , 0
  4450.7     .05       0  4986.5     .05       0  5010.6     .05       0
Bank Sta=4986.5,5010.6
XS Rating Curve= 0 ,0
Exp/Cntr=0.3,0.1

Type RM Length L Ch R = 1 ,70000   ,500,500,500
BEGIN DESCRIPTION:
PECAN CREEK 140.0
END DESCRIPTION:
XS GIS Cut Line= 3
      2796055.69     10292953.13      2795953.36     10292529.41
      2795455.66     10292053.09
#Sta/Elev= 30
  4564.1 1357.91  4582.5 1354.36  4636.1 1338.79  4656.7 1334.91  4677.3 1327.93
  4697.9 1325.72  4718.4 1320.37  4760.3 1313.94  4790.4 1311.25  4913.9 1308.22
  4964.5 1304.52  4983.5 1301.39    4984 1300.89  5007.6 1301.39  5031.1    1303
  5059.4 1307.87  5087.7 1306.51    5116 1309.49  5151.2 1309.05  5179.5 1311.86
  5271.7  1316.3  5335.2 1317.05  5377.7 1320.56  5412.9 1319.17  5476.7 1325.94
  5526.1 1338.36  5596.9 1348.79  5618.3 1353.83  5674.9 1355.49  5688.9 1354.29
#Mann= 3 ,-1 , 0
  4564.1     .05       0  4983.5     .05       0  5007.6     .05       0
Bank Sta=4983.5,5007.6
XS Rating Curve= 0 ,0
Exp/Cntr=0.3,0.1

Type RM Length L Ch R = 1 ,69500   ,500,500,500
BEGIN DESCRIPTION:
PECAN CREEK 139.0
END DESCRIPTION:
XS GIS Cut Line= 3
      2796255.65     10292003.12      2796010.99     10292050.46
       2795505.7     10292003.11
#Sta/Elev= 30
  4750.8 1315.83  4771.1 1314.84  4776.7 1315.61  4781.7 1314.27  4791.5 1313.82
  4811.9 1316.03  4828.4 1316.24  4833.5 1314.68  4842.4 1314.51  4852.6 1312.68
  4880.2  1305.3  4937.1 1302.69  4983.8 1294.15  4988.9 1294.79    4993 1293.43
  4993.5 1292.93  5017.6 1293.43  5045.5 1295.14  5095.7 1301.18  5176.1 1304.93
  5206.2  1309.5  5240.5 1311.23  5246.4 1312.58  5276.5 1314.72  5344.3  1318.2
  5366.9 1317.99  5417.1 1330.82  5437.2 1337.94  5467.3  1340.8  5507.5 1349.87
#Mann= 3 ,-1 , 0
  4750.8     .05       0    4993     .05       0  5017.6     .05       0
Bank Sta=4993,5017.6
XS Rating Curve= 0 ,0
Exp/Cntr=0.3,0.1

Type RM Length L Ch R = 1 ,69000   ,500,500,500
BEGIN DESCRIPTION:
PECAN CREEK 138.0
END DESCRIPTION:
XS GIS Cut Line= 3
      2796405.67     10291703.11      2796168.17     10291622.21
      2795955.72     10291553.12
#Sta/Elev= 30
  4749.1 1322.78  4796.1 1321.41  4822.2 1317.61  4827.5 1319.39  4833.6 1317.15
  4853.5 1314.62  4858.8  1316.4  4865.3 1312.99  4884.9 1309.09  4890.2 1309.96
  4907.5 1304.19  4928.7 1300.63  4966.7 1284.66  4967.2 1284.16  4991.3 1284.66
  5015.8 1285.83  5023.6 1287.91  5039.4 1288.99  5065.7 1295.48  5079.7 1301.08
  5097.3 1300.64  5106.4 1303.03  5111.6 1302.46  5138.3 1311.78  5143.6  1311.5
  5149.8 1315.57  5170.3 1321.01  5181.4  1320.4  5191.9 1322.91  5223.4 1323.54
#Mann= 3 ,-1 , 0
  4749.1     .05       0  4966.7     .05       0  4991.3     .05       0
Bank Sta=4966.7,4991.3
XS Rating Curve= 0 ,0
Exp/Cntr=0.3,0.1

Type RM Length L Ch R = 1 ,68500   ,500,500,500
BEGIN DESCRIPTION:
PECAN CREEK 137.0
END DESCRIPTION:
XS GIS Cut Line= 3
      2796655.69     10291453.12      2796408.34     10291185.52
      2795905.68     10290703.11
#Sta/Elev= 30
  4635.6 1337.12  4656.9 1336.74  4677.9 1329.44  4685.2 1328.68    4692 1324.74
  4756.1 1306.14  4762.9  1307.3  4770.3 1303.85  4840.6 1295.29    4848 1296.84
  4854.8 1295.11  4876.3 1294.54  4897.3 1289.87  4975.5 1285.25  4977.4 1281.69
  4977.9 1281.19    5002 1281.69    5039 1285.23  5077.9  1286.3  5180.5 1283.87
  5187.4 1286.75  5237.1 1291.49  5258.2 1295.89  5314.8 1303.14  5406.6 1312.19
  5489.8 1315.13  5569.5 1314.22  5590.6 1316.88  5597.8 1316.42  5696.7 1329.47
#Mann= 5 ,-1 , 0
  4635.6     .05       0  4977.4     .05       0    5002     .05       0
  5077.9     .12       0  5489.8     .05       0
Bank Sta=4977.4,5002
XS Rating Curve= 0 ,0
Exp/Cntr=0.3,0.1

Type RM Length L Ch R = 1 ,68000   ,500,500,500
BEGIN DESCRIPTION:
PECAN CREEK 136.0
END DESCRIPTION:
XS GIS Cut Line= 3
      2796905.68     10290953.11        2796525.     10290700.44
      2796305.65      10290653.1
#Sta/Elev= 30
  4543.1 1330.68  4607.7  1316.6  4622.8 1314.79  4628.8  1312.1  4664.9 1304.73
  4673.9 1304.55  4723.1 1296.21  4729.3 1296.06  4746.1 1294.52  4752.1 1296.53
  4767.1 1294.22  4773.1 1294.42  4803.2 1289.41  4809.2 1289.49  4818.3 1286.95
  4854.3 1281.09  4875.4 1285.15  4911.5 1287.01  4953.6 1287.13  4959.8 1285.59
  4968.6 1284.64  4983.4 1279.13  4983.9 1278.63  5009.8 1279.13    5030 1281.46
  5070.9 1279.47  5118.3 1287.39    5163 1294.99  5199.7 1299.91  5224.4 1301.66
#Mann= 6 ,-1 , 0
  4543.1     .12       0  4729.3     .05       0  4959.8     .12       0
  4983.4     .07       0  5009.8     .12       0  5118.3     .05       0
Bank Sta=4983.4,5009.8
XS Rating Curve= 0 ,0
Exp/Cntr=0.3,0.1

Type RM Length L Ch R = 1 ,67500   ,500,500,500
BEGIN DESCRIPTION:
PECAN CREEK 135.0
END DESCRIPTION:
XS GIS Cut Line= 3
      2796705.67     10290153.12      2796584.74     10290218.76
      2796255.68     10290303.11
#Sta/Elev= 30
  4862.4 1308.73  4870.5 1309.31  4885.1 1307.21  4892.3 1304.34    4898 1304.08
  4907.9 1301.29  4914.2 1296.08  4930.4 1290.72    4936 1286.76    4942 1283.74
  4957.9 1278.96  4979.8 1276.14  4982.7 1273.35  4983.2 1272.85  5009.2 1273.35
  5009.4 1274.83  5019.7 1275.79  5041.6    1275  5050.6 1273.65  5071.3 1274.34
  5112.6 1277.41  5143.6 1276.66  5153.6 1279.03  5158.8 1278.33  5164.2 1280.08
  5199.5 1284.23  5215.8  1287.5  5275.9 1296.65  5321.9 1302.66  5339.7 1303.92
#Mann= 3 ,-1 , 0
  4862.4     .12       0  4982.7     .07       0  5009.2     .12       0
Bank Sta=4982.7,5009.2
XS Rating Curve= 0 ,0
Exp/Cntr=0.3,0.1

Type RM Length L Ch R = 1 ,67000   ,500,500,500
BEGIN DESCRIPTION:
PECAN CREEK 134.0
END DESCRIPTION:
XS GIS Cut Line= 3
      2796805.67     10289853.11      2796404.52     10289756.16
      2796055.64     10289853.12
#Sta/Elev= 30
  4587.3 1310.29  4599.4 1308.77  4605.6 1306.46  4659.3 1299.12  4701.9 1296.68
    4715 1295.82  4736.4 1295.49  4778.2 1290.54  4783.4 1291.63  4820.1 1288.44
  4825.2 1289.88  4854.8 1288.94  4875.3 1285.74  4903.8 1277.43    4909 1277.96
  4917.4 1276.51  4957.6 1275.46  4987.5 1269.25  4997.5 1269.12    4998 1268.62
  5024.1 1269.12  5029.9 1270.67  5045.1 1270.94  5079.3 1275.32  5105.6 1276.54
  5164.6  1281.8  5192.4  1285.5  5271.3 1291.64  5305.5  1295.9  5362.1 1299.76
#Mann= 9 ,-1 , 0
  4587.3     .05       0  4599.4     .12       0  4701.9     .05       0
    4715     .12       0  4917.4     .05       0  4997.5     .05       0
  5024.1     .05       0  5105.6     .12       0  5164.6     .05       0
Bank Sta=4997.5,5024.1
XS Rating Curve= 0 ,0
Exp/Cntr=0.3,0.1

Type RM Length L Ch R = 1 ,66500   ,500,500,500
BEGIN DESCRIPTION:
PECAN CREEK 133.0
END DESCRIPTION:
XS GIS Cut Line= 3
      2796705.71     10289353.12      2796324.96     10289263.74
      2796105.69     10289203.11
#Sta/Elev= 30
  4608.9 1294.66  4717.6 1286.57    4760 1283.92  4765.1 1284.07  4773.3 1282.23
  4810.3 1279.68  4824.6 1277.76    4850 1276.42  4855.5  1275.5  4869.6  1275.1
  4927.4 1272.43  4958.2 1267.96  4977.2 1267.17  4983.8 1265.79  4984.3 1265.29
  5009.9 1265.29  5010.4 1265.79    5018  1267.3  5040.8 1267.26  5057.5  1273.4
  5062.7 1273.04  5071.9 1276.62  5082.3 1279.66  5091.8 1281.55    5103 1282.94
  5154.9 1286.57  5170.8 1284.95    5176 1285.58  5201.6 1285.66  5227.5 1288.41
#Mann= 5 ,-1 , 0
  4608.9     .05       0  4810.3     .12       0  4869.6     .05       0
  4983.8     .03       0  5010.4     .05       0
Bank Sta=4983.8,5010.4
XS Rating Curve= 0 ,0
Exp/Cntr=0.3,0.1

Type RM Length L Ch R = 1 ,66000   ,500,500,500
BEGIN DESCRIPTION:
PECAN CREEK 132.0
END DESCRIPTION:
XS GIS Cut Line= 3
      2796705.68     10289003.11      2796325.21     10288764.69
      2796255.68      10288253.1
#Sta/Elev= 30
    4551 1285.16  4616.4 1282.74  4634.5 1280.84  4680.8 1277.29    4726 1277.08
  4753.1 1274.75  4856.8 1271.23  4894.8 1267.88  4910.7 1265.62    4957 1264.69
    4964 1265.69  4972.3 1264.17  4978.2 1264.93  4996.8 1262.89  5011.7 1264.24
  5058.6 1263.12  5082.3  1263.3  5092.4 1262.88  5094.4 1261.69  5094.9 1261.19
    5121 1261.69  5122.7 1263.87  5142.9 1267.97  5173.2 1271.38  5233.7 1287.36
  5274.1 1290.33  5314.4 1300.19  5341.3 1298.29  5395.2 1302.12  5516.3 1314.09
#Mann= 8 ,-1 , 0
    4551     .12       0  4634.5     .05       0  4894.8     .12       0
  4910.7     .05       0  5058.6     .12       0  5094.4     .05       0
    5121     .12       0  5341.3     .05       0
Bank Sta=5094.4,5121
XS Rating Curve= 0 ,0
Exp/Cntr=0.3,0.1

Type RM Length L Ch R = 1 ,65500   ,500,500,500
BEGIN DESCRIPTION:
PECAN CREEK 131.0
END DESCRIPTION:
XS GIS Cut Line= 3
      2797055.71     10288753.13      2796666.98     10288517.63
      2796455.71     10288453.12
#Sta/Elev= 30
  4545.5  1290.3  4574.6 1288.31  4580.6 1287.09  4611.5 1284.69  4632.8 1282.11
  4662.5 1280.18  4675.5 1278.31  4770.5 1272.75  4822.8 1271.51  4865.5 1266.95
  4872.9 1267.64    4881 1267.27  4902.4 1264.79  4908.2 1262.25  4917.8 1260.82
  4939.2    1261    4953 1259.78  4953.5 1259.28  4979.3 1259.28  4979.8 1259.78
  5053.6 1261.27  5074.5 1269.81    5085 1270.47  5095.5 1272.34  5100.9 1274.28
  5126.8 1278.12  5138.9 1281.02  5179.1  1287.4  5205.4 1289.16  5220.9 1291.18
#Mann= 4 ,-1 , 0
  4545.5     .05       0    4953     .03       0  4979.8     .05       0
  5205.4     .12       0
Bank Sta=4953,4979.8
XS Rating Curve= 0 ,0
Exp/Cntr=0.3,0.1

Type RM Length L Ch R = 1 ,65000   ,321,321,321
BEGIN DESCRIPTION:
PECAN CREEK 130.0
END DESCRIPTION:
XS GIS Cut Line= 3
      2797155.68      10288353.1      2797072.47     10288248.07
      2796705.69     10287903.12
#Sta/Elev= 30
    4866 1281.15  4879.6 1280.58  4887.6 1281.58  4892.2 1280.58  4908.4 1279.25
  4929.8 1274.36  4958.1 1257.88  4966.2 1255.06  4967.2 1251.56  4967.7 1251.06
    4994 1251.56    5000 1253.04  5015.4 1254.35  5022.7 1258.16  5029.5 1260.06
  5043.7 1261.59  5057.8 1262.46  5100.3 1262.77  5107.2 1262.18    5178  1265.8
  5199.5  1269.5  5206.3 1268.93  5256.1 1273.18  5340.7 1276.89  5425.6 1284.09
  5461.2 1287.81  5489.6 1294.18  5496.4 1296.21  5500.1 1298.53  5503.5 1298.53
#Mann= 4 ,-1 , 0
    4866     .12       0  4892.2     .05       0  4967.2     .05       0
    4994     .05       0
Bank Sta=4967.2,4994
XS Rating Curve= 0 ,0
Exp/Cntr=0.3,0.1

Type RM Length L Ch R = 1 ,64679   ,679,679,679
BEGIN DESCRIPTION:
Mapping XS 37a18cbe
END DESCRIPTION:
XS GIS Cut Line= 3
      2797332.86     10288255.18      2797138.42     10287720.46
      2796242.56     10287817.68
#Sta/Elev= 30
  4712.6 1275.66  4780.7 1275.09  4861.9 1271.99  4885.1 1269.98  4903.1 1263.58
  4953.6 1251.56  4996.1 1250.24  4996.6 1249.74  5022.9 1250.24  5040.1 1251.51
  5045.4 1254.26  5065.4 1255.43  5070.7 1257.86    5096 1259.53  5101.3  1261.3
  5126.6 1260.22  5166.2  1263.7  5218.3 1267.85  5278.3 1281.99  5336.8 1281.23
  5436.6 1281.01  5455.3 1281.29  5495.6 1278.42  5536.5 1279.48  5636.3 1288.61
  5676.6    1293  5827.5 1300.78  6002.4 1305.04  6058.9 1303.68  6182.7 1310.06
#Mann= 9 ,-1 , 0
  4712.6     .05       0  4903.1     .12       0  4996.1     .07       0
  5022.9     .12       0  5166.2     .05       0  5336.8     .12       0
  5436.6     .05       0  5536.5     .12       0  5636.3     .05       0
Bank Sta=4996.1,5022.9
XS Rating Curve= 0 ,0
Exp/Cntr=0.3,0.1

Type RM Length L Ch R = 1 ,64000   ,500,500,500
BEGIN DESCRIPTION:
PECAN CREEK 128.0
END DESCRIPTION:
XS GIS Cut Line= 3
      2797455.72     10288053.09      2797642.96     10287935.88
       2797927.1      10287637.4
#Sta/Elev= 30
  4779.1  1268.7    4838 1265.79  4859.8  1263.1  4873.4 1263.24    4881 1260.98
  4896.3 1258.87  4902.2 1259.42  4917.6 1255.46  4923.5 1255.38  4938.8 1250.66
  4981.2 1245.45  4983.1 1243.64  4983.6 1243.14  5009.9 1243.64  5025.1 1244.71
  5036.7 1248.77  5067.6 1259.74  5074.5 1263.72  5081.7 1264.41  5088.6 1269.09
  5095.9 1270.14  5102.8 1275.04    5110 1276.94  5116.9 1281.06  5124.2 1283.52
  5159.4 1290.47    5195 1294.72  5244.3 1297.61    5322 1296.54  5412.1 1289.52
#Mann= 4 ,-1 , 0
  4779.1     .05       0  4983.1     .05       0  5009.9     .05       0
  5036.7     .12       0
Bank Sta=4983.1,5009.9
XS Rating Curve= 0 ,0
Exp/Cntr=0.3,0.1

Type RM Length L Ch R = 1 ,63500   ,500,500,500
BEGIN DESCRIPTION:
PECAN CREEK 127.0
END DESCRIPTION:
XS GIS Cut Line= 3
      2797355.71     10288403.11      2797687.15     10288431.98
       2797955.7     10288403.11
#Sta/Elev= 30
  4667.3 1275.16  4723.7 1270.54  4728.7  1270.7  4747.6 1269.02  4767.7 1266.32
  4905.2 1255.09  4928.3 1253.55  4948.3 1249.58  4954.4 1247.52  4959.4 1247.04
  4968.4 1244.72  4978.5 1244.19  4983.3 1243.28  4983.8 1242.78  5009.7 1242.78
  5010.2 1243.28  5018.6 1244.55    5040 1245.53  5048.8  1248.4  5058.9 1250.65
  5109.2 1257.35    5127 1261.29    5132 1261.11  5139.3 1263.45  5159.4 1267.27
  5186.9 1271.31  5209.7  1274.5  5224.1 1275.35  5259.9  1279.3  5270.1 1280.43
#Mann= 6 ,-1 , 0
  4667.3     .05       0  4905.2     .12       0  4983.3     .07       0
  5010.2     .12       0  5186.9     .05       0  5259.9     .12       0
Bank Sta=4983.3,5010.2
XS Rating Curve= 0 ,0
Exp/Cntr=0.3,0.1

Type RM Length L Ch R = 1 ,63000   ,500,500,500
BEGIN DESCRIPTION:
PECAN CREEK 126.0
END DESCRIPTION:
XS GIS Cut Line= 3
      2797355.65     10289003.13      2797577.48     10288908.41
      2797805.67     10288853.11
#Sta/Elev= 30
  4758.8 1274.36  4773.4 1273.61  4820.6 1266.54  4844.2 1263.61  4849.6 1263.91
  4873.2 1259.91  4889.3  1259.3  4896.8 1256.87  4902.3 1256.47  4920.4 1249.28
  4925.9  1250.7  4943.7 1244.24  4949.5 1241.18  4954.9 1242.32  4973.1 1239.26
    4995 1237.87  4995.5 1237.37  5021.9 1237.87    5029 1241.19  5049.4 1243.61
  5085.9 1249.87  5091.1 1248.42  5111.3 1251.26  5127.7 1254.72  5132.9 1253.51
  5152.1 1255.73  5169.5 1257.63  5174.7  1257.2  5203.9 1261.07  5234.8 1262.29
#Mann= 5 ,-1 , 0
  4758.8     .05       0    4995     .05       0  5021.9     .05       0
  5049.4     .12       0  5152.1     .05       0
Bank Sta=4995,5021.9
XS Rating Curve= 0 ,0
Exp/Cntr=0.3,0.1

Type RM Length L Ch R = 1 ,62500   ,500,500,500
BEGIN DESCRIPTION:
PECAN CREEK 125.0
END DESCRIPTION:
XS GIS Cut Line= 3
      2797305.64      10289353.1      2797530.09     10289401.93
      2797755.64     10289503.09
#Sta/Elev= 30
  4770.3 1263.48  4789.8 1260.96  4794.9 1261.39  4838.9 1254.43    4844 1254.79
  4882.9 1248.93    4888 1249.28  4893.2 1247.06  4903.4 1246.62  4937.1 1241.38
  4944.3 1238.98  4954.6 1238.03  4967.6 1235.42  4968.1 1234.92  4994.5 1235.42
  5018.8 1237.36  5028.1 1240.52  5065.2 1247.17  5071.9 1249.76  5082.8 1252.36
  5093.9 1256.77  5104.8  1258.8  5111.5 1260.91  5140.2 1265.06  5157.9 1266.92
  5186.6 1267.97  5203.4  1269.4  5232.9 1269.69  5238.4 1268.68  5247.2 1269.13
#Mann= 3 ,-1 , 0
  4770.3     .12       0  4967.6     .07       0  4994.5     .12       0
Bank Sta=4967.6,4994.5
XS Rating Curve= 0 ,0
Exp/Cntr=0.3,0.1

Type RM Length L Ch R = 1 ,62000   ,500,500,500
BEGIN DESCRIPTION:
PECAN CREEK 124.0
END DESCRIPTION:
XS GIS Cut Line= 3
      2796955.72     10289853.11       2797440.4     10289886.18
      2797705.66     10289703.13
#Sta/Elev= 30
  4514.2 1303.16  4544.2 1292.21  4564.3 1281.96  4583.5 1275.57  4654.5 1258.77
  4737.1 1250.87  4880.7 1243.61  4935.1 1239.18  4945.2 1236.21  4955.2 1235.35
  4985.3 1235.11    4993 1232.81  4993.5 1232.31  5019.9 1232.81  5028.2 1236.95
  5034.3 1236.84  5049.2 1240.82  5055.3 1239.75  5070.1 1242.17  5078.9 1245.64
    5085 1245.16  5091.5 1248.22  5100.6 1249.71    5106 1248.57  5114.8 1250.71
  5120.8 1250.13  5150.6 1257.11  5224.6  1260.6  5279.1 1261.03  5322.3 1259.04
#Mann= 5 ,-1 , 0
  4514.2     .05       0    4993     .05       0  5019.9     .05       0
  5100.6     .12       0  5224.6     .05       0
Bank Sta=4993,5019.9
XS Rating Curve= 0 ,0
Exp/Cntr=0.3,0.1

Type RM Length L Ch R = 1 ,61500   ,500,500,500
BEGIN DESCRIPTION:
PECAN CREEK 123.0
END DESCRIPTION:
XS GIS Cut Line= 3
      2797405.68     10290553.11      2797431.21     10290323.72
      2797705.67     10289803.14
#Sta/Elev= 30
  4769.2 1295.85  4789.3 1293.53  4814.4 1292.56  4839.6 1288.88  4879.9 1279.82
  4899.9 1272.42  4904.9  1273.4  4910.1 1269.47  4970.4 1237.72  4980.5 1233.29
  4984.3 1230.21  4984.8 1229.71  5011.2 1230.21    5019 1231.58    5063 1235.39
  5107.1 1235.71  5129.1 1238.81  5167.5 1239.88  5193.5 1241.73  5255.2 1244.53
    5316  1249.1  5321.7 1248.23  5338.1 1250.94  5441.6 1252.84  5448.2 1252.28
  5464.2 1252.88  5470.2 1254.15  5492.2 1253.62  5543.3 1255.15  5588.5 1255.06
#Mann= 5 ,-1 , 0
  4769.2     .12       0  4984.3     .07       0  5011.2     .12       0
  5193.5     .12       0  5255.2     .05       0
Bank Sta=4984.3,5011.2
XS Rating Curve= 0 ,0
Exp/Cntr=0.3,0.1

Type RM Length L Ch R = 1 ,61000   ,500,500,500
BEGIN DESCRIPTION:
PECAN CREEK 122.0
END DESCRIPTION:
XS GIS Cut Line= 3
      2798359.46     10290485.02      2797881.01     10290161.97
      2797705.68     10289803.11
#Sta/Elev= 30
  4422.7 1284.04  4449.1 1282.04  4455.2 1283.53  4470.1 1280.62  4476.2 1282.89
  4506.1 1278.77  4527.1 1281.48  4542.1 1278.59  4563.1 1280.17    4572 1279.01
    4578 1281.43    4593 1275.96    4614 1274.94    4629 1271.12    4650 1271.99
    4665 1267.01    4686 1266.94  4700.9 1263.39  4721.9 1262.32  4765.1 1255.18
  4808.8 1252.17  4814.9 1254.65  4838.4 1251.21  4967.7 1230.61  5028.1 1228.45
  5028.6 1227.95  5055.8 1228.45  5092.1 1235.47  5121.2 1239.49  5399.4 1255.06
#Mann= 5 ,-1 , 0
  4422.7     .05       0  4838.4     .12       0  5028.1     .07       0
  5055.8     .12       0  5092.1     .05       0
Bank Sta=5028.1,5055.8
XS Rating Curve= 0 ,0
Exp/Cntr=0.3,0.1
