--- SAND SPRING CREEK.prj (project) ---

Proj Title=SAND SPRING CREEK Base Level Engineering
Current Plan=p01
Default Exp/Contr=0.3,0.1
English Units
Geom File=g01
Flow File=f01
Plan File=p01
Y Axis Title=Elevation
X Axis Title(PF)=Main Channel Distance
X Axis Title(XS)=Station
BEGIN DESCRIPTION:
SAND SPRING CREEK
END DESCRIPTION:
DSS Export Rating Curves= 0
DSS Export Rating Curve Sorted= 0
DSS Export Volume Flow Curves= 0
DXF OffsetX= 0
DXF OffsetY= 0
DXF ScaleX= 1
DXF ScaleY= 10

--- SAND SPRING CREEK.p01 (plan) ---

Plan Title=Multiple Run
Short Identifier=Multiple
Geom File=g01
Flow File=f01
Subcritical Flow
K Sum by GR= 0
Std Step Tol= 0.01
Critical Tol= 0.01
Num of Std Step Trials= 20
Max Error Tol= 0.3
Flow Tol Ratio= 0.001
Split Flow NTrial= 30
Split Flow Tol= 0.02
Split Flow Ratio= 0.02
Log Output Level= 0
Friction Slope Method= 1
Unsteady Friction Slope Method= 2
Unsteady Bridges Friction Slope Method= 1
Parabolic Critical Depth
Global Vel Dist=  1 , 1 , 1
Global Log Level= 0
CheckData=True
Encroach Param= -1, 0, 0, 0
BEGIN DESCRIPTION:
Multiple Run
END DESCRIPTION:

--- SAND SPRING CREEK.f01 (steady flow) ---

Flow Title=Multiple
Number of Profiles=7
Profile Names=10-year,25-year,50-year,1pct_min,100-year,1pct_plu,500-year
River Rch & RM= SAND SPRING CREE,Reach-1,40500
     477     775    1676    1234    2374    4567    3465
River Rch & RM= SAND SPRING CREE,Reach-1,31500
     809    1369    2778    1734    3976    9117    5752
River Rch & RM= SAND SPRING CREE,Reach-1,24000
    1135    1966    4018    2510    5816   13480    8401
River Rch & RM= SAND SPRING CREE,Reach-1,17500
    1358    2379    4905    4072    7141   12523   10292
River Rch & RM= SAND SPRING CREE,Reach-1,14000
    1678    2986    5910    4955    8627   15019   12373
River Rch & RM= SAND SPRING CREE,Reach-1,7500
    1939    3497    6578    5058    9608   18250   13736
Boundary for River Rch & Prof#=SAND SPRING CREE,Reach-1,1
Up Type=0
Dn Type=3
Dn Slope=0.005
Boundary for River Rch & Prof#=SAND SPRING CREE,Reach-1,2
Up Type=0
Dn Type=3
Dn Slope=0.005
Boundary for River Rch & Prof#=SAND SPRING CREE,Reach-1,3
Up Type=0
Dn Type=3
Dn Slope=0.005
Boundary for River Rch & Prof#=SAND SPRING CREE,Reach-1,4
Up Type=0
Dn Type=3
Dn Slope=0.005
Boundary for River Rch & Prof#=SAND SPRING CREE,Reach-1,5
Up Type=0
Dn Type=3
Dn Slope=0.005
Boundary for River Rch & Prof#=SAND SPRING CREE,Reach-1,6
Up Type=0
Dn Type=3
Dn Slope=0.005
Boundary for River Rch & Prof#=SAND SPRING CREE,Reach-1,7
Up Type=0
Dn Type=3
Dn Slope=0.005

--- SAND SPRING CREEK.g01 (geometry) ---

Geom Title=Existing Conditions
Program Version=4.10

River Reach=SAND SPRING CREE,Reach-1
Reach XY= 30
      2773084.25       10296265.      2771932.25       10294506.
       2772288.5       10292454.        2772181.       10290516.
        2771634.       10290426.        2770202.       10288375.
      2768949.75       10287390.      2769207.25       10286300.
      2768802.75       10285711.      2769795.75       10284805.
        2770111.       10283049.      2771128.25       10281233.
        2771789.       10280761.      2771682.25       10280004.
      2773463.75       10278923.       2773689.5       10277789.
        2776311.       10275039.       2776170.5       10274541.
        2776929.       10273846.       2776288.5       10273251.
        2777127.       10272746.      2777786.75       10271242.
      2777989.75       10270286.        2777778.       10270114.
      2778519.25       10268761.      2778260.75       10268253.
      2778418.75       10267499.       2779170.5       10266935.
      2779777.25       10267266.      2780326.25       10267064.

Type RM Length L Ch R = 1 ,40500   ,500,500,500
BEGIN DESCRIPTION:
SAND SPRING CREEK 80.0
END DESCRIPTION:
XS GIS Cut Line= 3
      2773455.64     10296303.08      2773069.82     10296039.09
      2772705.66     10296453.13
#Sta/Elev= 30
  4532.5 1573.45  4590.7 1569.32  4607.9 1569.41  4713.3 1566.66  4770.1 1562.85
  4858.7 1561.21  4907.6 1558.93  4928.6 1556.33  4949.5 1556.31  4964.5 1553.94
  4985.4 1553.24  4997.5 1550.29  4997.7 1549.79  5001.5 1550.29  5041.4 1551.79
    5048 1554.64  5055.6 1553.58  5062.3 1555.49  5069.8  1554.3  5084.1 1555.12
  5119.2 1559.01    5197 1562.45  5211.2  1564.8  5225.5 1564.28  5304.3 1569.91
  5360.2 1573.19  5465.3 1585.48  5473.1 1584.88  5544.3 1593.47  5551.4 1595.32
#Mann= 7 ,-1 , 0
  4532.5     .05       0  4607.9     .12       0  4858.7     .05       0
  4997.5     .05       0  5001.5     .05       0  5304.3     .12       0
  5465.3     .05       0
Bank Sta=4997.5,5001.5
XS Rating Curve= 0 ,0
Exp/Cntr=0.3,0.1

Type RM Length L Ch R = 1 ,40000   ,500,500,500
BEGIN DESCRIPTION:
SAND SPRING CREEK 79.0
END DESCRIPTION:
XS GIS Cut Line= 3
      2773255.71     10295153.08      2772851.83     10295637.63
      2772355.71     10296053.09
#Sta/Elev= 30
  4369.2 1630.88  4372.5 1630.88  4440.2 1611.78  4454.5 1606.43    4461 1605.59
  4483.1 1598.46  4546.9 1581.93  4633.4 1562.87  4660.2 1557.18  4674.5 1556.46
  4688.8 1553.62  4824.2 1547.34  4851.5 1543.85  4873.6 1544.51  4958.3 1540.92
  4966.1 1541.81  5015.4 1540.52  5036.3 1541.78  5120.1 1540.46  5120.4 1539.96
  5124.1 1540.46  5157.3 1542.71  5214.4 1543.03  5306.7 1546.69  5327.7 1547.63
  5356.3 1546.71  5391.5 1549.86  5512.8 1555.25  5558.3  1558.3  5647.1 1563.11
#Mann= 8 ,-1 , 0
  4369.2     .12       0  4633.4     .05       0  5120.1     .05       0
  5124.1     .05       0  5214.4     .12       0  5306.7     .05       0
  5512.8     .12       0  5558.3     .05       0
Bank Sta=5120.1,5124.1
XS Rating Curve= 0 ,0
Exp/Cntr=0.3,0.1

Type RM Length L Ch R = 1 ,39500   ,500,500,500
BEGIN DESCRIPTION:
SAND SPRING CREEK 78.0
END DESCRIPTION:
XS GIS Cut Line= 3
      2772855.66     10294853.14      2772478.75     10295342.52
      2771955.66     10295753.13
#Sta/Elev= 30
  4382.3 1616.76  4389.5 1616.65  4395.8 1612.17  4439.3 1600.48  4445.6 1596.15
  4453.8 1595.39  4460.2 1591.22  4468.3 1590.26  4489.2 1581.19  4503.7 1579.58
  4538.4 1567.73  4588.8 1554.65  4603.3 1553.32  4624.1 1545.72  4688.5 1531.86
  4704.2 1531.01  4799.6 1527.54    4865 1526.92  4865.2 1526.42    4869 1526.92
  5087.4 1530.56  5386.6  1541.9  5409.1 1539.45    5487 1538.89  5494.1 1542.48
  5537.5 1547.13  5543.8 1550.17  5587.2 1550.32  5628.8 1547.11    5665 1550.79
#Mann= 7 ,-1 , 0
  4382.3     .12       0  4538.4     .05       0  4704.2     .12       0
  4799.6     .05       0    4865     .05       0    4869     .05       0
  5087.4     .12       0
Bank Sta=4865,4869
XS Rating Curve= 0 ,0
Exp/Cntr=0.3,0.1

Type RM Length L Ch R = 1 ,39000   ,500,500,500
BEGIN DESCRIPTION:
SAND SPRING CREEK 77.0
END DESCRIPTION:
XS GIS Cut Line= 3
      2772705.64     10294703.13      2772289.43     10294902.97
      2771305.69     10295253.11
#Sta/Elev= 30
  4538.3 1576.24  4592.1 1559.06  4620.3 1553.86  4637.4 1547.72  4642.9 1547.57
  4649.2 1543.76  4704.6 1526.71  4733.5 1522.42  4778.1 1519.91  4801.4 1518.67
  4993.7 1518.65  5023.2 1516.27  5023.5 1515.77  5027.2 1516.27  5048.4 1517.99
  5162.6  1519.9  5208.3 1521.25  5269.3 1521.43  5436.4 1526.51  5556.7 1529.05
  5654.4 1533.65  5664.9 1533.29  5693.9 1533.35  5768.2    1540  5854.4 1552.26
  5874.4 1556.31  5879.9 1559.26  5910.8 1564.69    5998 1587.29  6044.2 1593.66
#Mann= 9 ,-1 , 0
  4538.3     .12       0  4778.1     .05       0  5023.2     .05       0
  5027.2     .05       0  5162.6     .12       0  5208.3     .05       0
  5436.4     .12       0  5654.4     .05       0  5664.9     .12       0
Bank Sta=5023.2,5027.2
XS Rating Curve= 0 ,0
Exp/Cntr=0.3,0.1

Type RM Length L Ch R = 1 ,38500   ,500,500,500
BEGIN DESCRIPTION:
SAND SPRING CREEK 76.0
END DESCRIPTION:
XS GIS Cut Line= 3
      2772755.65     10294603.11      2771943.26     10294545.89
      2771455.66     10294953.13
#Sta/Elev= 30
  4185.6 1597.99  4188.1 1597.99  4195.6 1593.36  4235.7 1577.39  4275.8  1563.4
  4295.8 1557.85    4346 1546.95  4386.1 1535.73  4395.1  1532.1  4400.1 1531.86
  4406.1 1528.71  4426.2 1524.27  4436.2 1522.24  4476.3 1518.61  4568.7 1513.61
  4586.6 1512.57  4807.1 1510.82  4857.2 1511.75  5015.7 1509.06    5016 1508.56
  5019.7 1509.06  5379.5 1520.63  5408.2 1519.41    5429 1521.63  5471.9 1523.13
  5478.9 1524.86  5543.5 1529.33  5586.9 1533.84  5615.4 1537.16  5635.3 1539.03
#Mann= 6 ,-1 , 0
  4185.6     .12       0  4568.7     .05       0  5015.7     .05       0
  5019.7     .05       0  5586.9     .12       0  5615.4     .05       0
Bank Sta=5015.7,5019.7
XS Rating Curve= 0 ,0
Exp/Cntr=0.3,0.1

Type RM Length L Ch R = 1 ,38000   ,500,500,500
BEGIN DESCRIPTION:
SAND SPRING CREEK 75.0
END DESCRIPTION:
XS GIS Cut Line= 3
      2772905.66      10294603.1      2771941.95      10294086.8
      2770955.72     10294753.08
#Sta/Elev= 30
  3906.7 1635.19  3952.1    1634  3974.7 1630.03  3996.9 1623.37  4031.5 1606.87
  4046.4 1601.78  4068.3 1590.12  4134.1 1565.76  4156.3 1558.67  4188.6 1553.21
  4232.4 1540.53  4254.4 1537.14    4282 1528.95  4380.3 1518.77  4492.3 1512.99
  4644.1 1505.04  4991.7 1499.13  4991.9 1498.63  4995.7 1499.13  5224.8 1503.92
  5319.6 1502.56  5427.5 1504.49  5671.3 1514.26  5808.1 1517.74  5906.9 1522.84
  5960.9 1527.07  6002.9 1535.69  6125.8  1563.9  6167.8  1579.3  6190.2 1583.98
#Mann= 5 ,-1 , 0
  3906.7     .12       0  4492.3     .05       0  4991.7     .05       0
  4995.7     .05       0  5906.9     .12       0
Bank Sta=4991.7,4995.7
XS Rating Curve= 0 ,0
Exp/Cntr=0.3,0.1

Type RM Length L Ch R = 1 ,37500   ,500,500,500
BEGIN DESCRIPTION:
SAND SPRING CREEK 74.0
END DESCRIPTION:
XS GIS Cut Line= 3
      2772555.67      10294053.1      2772153.33     10293674.73
      2770724.21     10293569.39
#Sta/Elev= 30
  4447.7 1514.13  4454.8 1513.06  4617.4 1505.13  4638.9 1503.23    4653 1503.44
  4694.8    1501  4836.7 1494.09  4921.7 1491.14  4935.8 1491.41  4956.9 1490.11
  5077.9  1491.8  5178.1  1489.8  5218.2 1490.77  5308.5 1490.58  5362.9 1491.51
  5468.9 1490.62  5649.9 1491.34  5653.4 1491.27  5739.6 1488.96  5837.9 1488.23
  5838.2 1487.73  5841.9 1488.23    5860 1489.01  5910.7 1488.84  6020.4 1492.08
  6043.9 1491.41  6130.7 1493.65  6341.3 1503.13  6361.3 1505.01    6433 1508.55
#Mann= 6 ,-1 , 0
  4447.7     .12       0  4694.8     .05       0  5649.9     .12       0
  5653.4     .05       0  5837.9     .05       0  5841.9     .05       0
Bank Sta=5837.9,5841.9
XS Rating Curve= 0 ,0
Exp/Cntr=0.3,0.1

Type RM Length L Ch R = 1 ,37000   ,500,500,500
BEGIN DESCRIPTION:
SAND SPRING CREEK 73.0
END DESCRIPTION:
XS GIS Cut Line= 3
      2773055.71     10293853.13      2772130.65     10293205.19
      2770866.46     10293284.88
#Sta/Elev= 30
  3870.6 1617.21  3907.3 1609.66  3934.7 1598.22  3949.5  1594.5  3964.3 1585.47
  3985.3 1577.79  4000.1 1570.02  4029.3  1560.9  4035.8 1556.68  4056.8 1548.76
  4078.2 1545.09  4092.5 1546.56  4101.2 1541.09  4122.1 1532.97  4200.3 1515.63
  4275.7 1509.11  4416.8 1499.88  4717.6 1484.97  4894.3 1480.03  4894.6 1479.53
  4898.3 1480.03  5475.9 1485.36  5656.3 1484.09  5676.3  1485.1  5686.8 1487.81
  5716.4 1482.79  5766.5 1483.29  5816.6 1488.12  6147.2  1503.1  6266.7 1512.18
#Mann= 4 ,-1 , 0
  3870.6     .12       0  4275.7     .05       0  4894.3     .05       0
  4898.3     .05       0
Bank Sta=4894.3,4898.3
XS Rating Curve= 0 ,0
Exp/Cntr=0.3,0.1

Type RM Length L Ch R = 1 ,36500   ,500,500,500
BEGIN DESCRIPTION:
SAND SPRING CREEK 72.0
END DESCRIPTION:
XS GIS Cut Line= 3
      2773155.69     10293703.12      2772203.47     10292730.28
      2771205.73     10292803.11
#Sta/Elev= 30
  3638.7 1589.34  3642.2 1589.34  3645.8 1584.22  3652.8 1584.51  3659.9 1581.96
  3666.9 1581.87  3674.1 1578.12  3681.1  1578.4  3688.2 1574.61  3695.2 1573.66
  3702.4 1569.36  3709.4 1568.99  3722.9  1564.6  3758.9 1552.85  3829.7 1538.39
  3879.1 1525.81  3928.7 1519.35  4147.8 1503.99  4395.3 1490.65  4706.5 1477.72
  4720.6 1476.19  4791.3 1475.75  4916.6 1471.87  4916.9 1471.37  4920.6 1471.87
  5228.4 1475.61  5383.1 1474.18  5428.9 1476.38  5649.5 1481.64  6000.4 1498.58
#Mann= 4 ,-1 , 0
  3638.7     .12       0  3722.9     .05       0  4916.6     .05       0
  4920.6     .05       0
Bank Sta=4916.6,4920.6
XS Rating Curve= 0 ,0
Exp/Cntr=0.3,0.1

Type RM Length L Ch R = 1 ,36000   ,500,500,500
BEGIN DESCRIPTION:
SAND SPRING CREEK 71.0
END DESCRIPTION:
XS GIS Cut Line= 3
      2773205.68     10293203.11      2772263.51     10292250.69
      2771255.67     10292303.11
#Sta/Elev= 30
  3660.3 1533.81  3663.8 1533.81  3674.4  1530.9  3688.5 1529.28  3705.9  1524.9
  3738.1 1519.03  3773.4 1509.45  3837.1 1502.73  3943.1 1497.89  3964.4 1496.13
  4247.2 1480.83  4544.2 1468.94  4643.2  1466.5    4820 1466.14  4897.8 1465.03
  4940.2 1465.44  4987.7 1464.42  4987.9 1463.92  4991.7 1464.42  4994.9 1465.03
  5017.8 1464.69  5087.9 1466.17    5128 1467.73    5143 1467.16  5258.2  1468.8
  5348.3 1468.13  5468.5 1471.61  5758.8 1482.71  5949.1  1492.1  6009.2 1495.88
#Mann= 4 ,-1 , 0
  3660.3     .12       0  3705.9     .05       0  4987.7     .05       0
  4991.7     .05       0
Bank Sta=4987.7,4991.7
XS Rating Curve= 0 ,0
Exp/Cntr=0.3,0.1

Type RM Length L Ch R = 1 ,35500   ,500,500,500
BEGIN DESCRIPTION:
SAND SPRING CREEK 70.0
END DESCRIPTION:
XS GIS Cut Line= 3
      2773555.66     10292903.09      2772269.65     10291765.73
       2771255.7      10292253.1
#Sta/Elev= 30
  3283.2 1512.42  3304.5 1517.83  3325.4 1517.85  3332.9 1521.33  3339.6 1519.34
  3347.2 1522.31  3353.8 1518.73  3361.4 1524.13  3368.1 1519.19  3375.6 1521.17
  3382.3 1517.17  3389.8 1518.47  3396.5 1513.44  3410.7 1513.73  3417.4 1509.94
  3439.2 1507.99  3460.1 1502.39  3552.1  1488.9  3899.2 1472.79  4097.5 1466.06
  4437.9 1460.79  4854.2 1459.58  4854.4 1459.08  4858.2 1459.58    4975 1460.16
  5123.9 1462.34  5337.3 1463.94  5607.4 1471.65  5952.5 1486.26    6125 1496.01
#Mann= 5 ,-1 , 0
  3283.2     .05       0  4854.2     .07       0  4858.2     .05       0
    4975     .12       0  5123.9     .05       0
Bank Sta=4854.2,4858.2
XS Rating Curve= 0 ,0
Exp/Cntr=0.3,0.1

Type RM Length L Ch R = 1 ,35000   ,184,184,184
BEGIN DESCRIPTION:
SAND SPRING CREEK 69.0
END DESCRIPTION:
XS GIS Cut Line= 3
       2773612.2      10292802.4      2772169.71     10291284.21
      2771155.69     10292103.11
#Sta/Elev= 30
  2905.8    1490  2909.9 1491.21  2917.1 1490.25    2924 1491.94  2931.3 1490.25
  2938.2 1491.37  2945.4 1489.47  2952.3 1490.08  3051.4 1483.78    3193 1479.26
  3242.3 1479.12  3383.9 1471.33  3617.3 1464.34  3864.8 1459.39    3985 1459.69
  4034.7 1457.96  4055.8 1459.14    4565 1457.95  4860.3 1455.72  4860.6 1455.22
  4864.3 1455.72  5200.8 1457.98  5343.1 1462.24  5642.2 1467.37  5819.7 1476.41
  5904.9 1478.98  6033.5  1486.6  6153.9 1491.61  6182.7 1491.42  6303.4 1499.45
#Mann= 3 ,-1 , 0
  2905.8     .05       0  4860.3     .05       0  4864.3     .05       0
Bank Sta=4860.3,4864.3
XS Rating Curve= 0 ,0
Exp/Cntr=0.3,0.1

Type RM Length L Ch R = 1 ,34816   ,316,316,316
BEGIN DESCRIPTION:
Mapping XS cc4775a7
END DESCRIPTION:
XS GIS Cut Line= 5
      2773336.49     10289715.59      2773174.84     10290316.93
      2772211.38     10291054.06      2772069.13     10291138.12
      2771449.55     10291712.53
#Sta/Elev= 30
  3060.9 1484.28  3099.8 1483.94  3118.5 1482.65  3238.4  1479.5  3410.4  1471.7
  3555.4 1463.05  3627.9 1461.04  3687.2 1457.06  3795.1 1455.59  3965.6 1450.93
  4065.3 1449.93  4079.8 1450.49  4115.2 1449.28  4227.4 1448.32  4227.7 1447.82
  4231.4 1448.32  4400.2 1449.47  4728.1 1455.47  4821.5 1454.55  4836.1 1453.55
  4938.2 1453.34    5075 1455.63  5145.9  1455.9  5336.9 1460.21  5499.7 1460.45
  5577.3 1462.19  5598.4 1461.46  5626.7    1463  5676.6 1463.87  5906.8 1473.63
#Mann= 3 ,-1 , 0
  3060.9     .05       0  4227.4     .05       0  4231.4     .05       0
Bank Sta=4227.4,4231.4
XS Rating Curve= 0 ,0
Exp/Cntr=0.3,0.1

Type RM Length L Ch R = 1 ,34500   ,500,500,500
BEGIN DESCRIPTION:
SAND SPRING CREEK 68.0
END DESCRIPTION:
XS GIS Cut Line= 3
      2772805.66     10289803.15      2772176.88      10290799.9
      2771305.65     10291753.14
#Sta/Elev= 30
  3821.5 1483.88  3847.6 1481.88  3905.9  1479.1  3938.5 1476.66  3951.5 1476.99
  3965.6 1475.26  4111.5  1467.9  4263.4 1461.07  4400.8 1456.99  4646.3 1452.48
  4691.1 1451.31  4753.5 1450.94  4753.8 1450.44  4757.5 1450.94    5034 1452.34
  5034.3 1452.33  5272.3 1453.62  5399.3 1456.41  5495.2 1456.97  5562.1 1458.17
  5604.7 1457.68  5640.4 1458.46    5649  1457.8  5696.5 1458.84  5710.7  1458.2
  5795.8 1458.91  5979.8 1465.11    6008 1465.17  6241.7 1474.75  6291.4 1478.01
#Mann= 11 ,-1 , 0
  3821.5     .05       0  3847.6     .12       0  3905.9     .05       0
  4646.3     .12       0  4691.1     .05       0  4753.5     .05       0
  4757.5     .05       0    5034     .12       0  5034.3     .05       0
  5495.2     .12       0    5649     .05       0
Bank Sta=4753.5,4757.5
XS Rating Curve= 0 ,0
Exp/Cntr=0.3,0.1

Type RM Length L Ch R = 1 ,34000   ,500,500,500
BEGIN DESCRIPTION:
SAND SPRING CREEK 67.0
END DESCRIPTION:
XS GIS Cut Line= 3
      2772805.69      10289603.1      2772009.88     10290440.05
      2771073.89     10291307.14
#Sta/Elev= 30
  3845.1 1496.94  3873.2 1496.04    3944  1488.9  4052.8 1482.48  4096.5  1480.3
  4241.3 1472.26  4446.4 1462.58  4755.5 1451.62  4851.3 1449.91  4904.2 1448.96
  4904.5 1448.46  4908.2 1448.96  4934.6 1450.05  5097.6 1449.88  5212.3 1450.16
  5507.7 1450.42  5755.5  1453.3  5811.6 1454.74  5889.9 1458.77  5910.8 1458.78
  5946.3 1461.16    6031 1462.96  6038.4 1464.12  6059.4 1463.57  6080.9 1464.95
  6130.3  1465.1  6201.1 1467.24  6207.9 1466.22  6236.3 1466.54  6275.9 1468.29
#Mann= 9 ,-1 , 0
  3845.1     .05       0  4052.8     .12       0  4096.5     .05       0
  4755.5     .12       0  4851.3     .05       0  4904.2     .05       0
  4908.2     .05       0  5097.6     .12       0  5212.3     .05       0
Bank Sta=4904.2,4908.2
XS Rating Curve= 0 ,0
Exp/Cntr=0.3,0.1

Type RM Length L Ch R = 1 ,33500   ,500,500,500
BEGIN DESCRIPTION:
SAND SPRING CREEK 66.0
END DESCRIPTION:
XS GIS Cut Line= 3
      2772505.66     10289353.14      2771573.61     10290352.98
      2771155.66     10290853.14
#Sta/Elev= 30
  3633.1 1490.35  3654.3 1490.47    3711 1488.31  3802.8 1482.27  3965.5 1473.97
  3972.9 1474.29  3979.7 1473.17    3987  1473.7  4043.2 1470.87  4050.5 1471.37
  4167.7 1465.14  4192.2 1464.43  4227.7 1461.77  4397.4 1454.31  4496.1 1451.03
  4630.9 1450.05  4687.1  1448.6  4913.8 1448.22  4961.1 1447.57  4961.4 1447.07
  4965.1 1447.57  4996.7 1447.75  5190.4 1450.46  5360.9 1456.88  5481.9 1459.26
  5488.4 1460.31  5517.1 1461.12  5523.6  1462.4  5609.5 1465.14  5651.8 1470.93
#Mann= 5 ,-1 , 0
  3633.1     .05       0  4167.7     .12       0  4227.7     .05       0
  4913.8     .07       0  4996.7     .05       0
Bank Sta=4961.1,4965.1
XS Rating Curve= 0 ,0
Exp/Cntr=0.3,0.1

Type RM Length L Ch R = 1 ,33000   ,500,500,500
BEGIN DESCRIPTION:
SAND SPRING CREEK 65.0
END DESCRIPTION:
XS GIS Cut Line= 3
      2772255.66     10289253.13      2771314.93     10289948.59
      2771055.68     10290903.12
#Sta/Elev= 30
  3830.1 1479.87  3872.9 1477.91  3887.5 1475.89  3958.4 1473.16  4309.2  1454.9
  4524.2 1448.94  4761.5 1446.56  4866.1 1446.16  4958.5 1444.21  4958.8 1443.71
  4962.5 1444.21  4974.2 1444.96  5004.9 1444.43  5132.4 1446.35  5263.7 1447.08
  5435.3 1451.79  5514.9 1452.38  5543.5 1454.32  5549.5 1453.41  5595.3 1457.26
  5623.9 1457.64  5629.1 1458.99  5702.9 1460.03  5738.2  1461.9  5750.8 1464.03
  5761.1 1463.93  5802.6  1467.1  5857.6 1467.57  5916.6 1471.06  5989.1  1472.6
#Mann= 5 ,-1 , 0
  3830.1     .05       0  4761.5     .12       0  4866.1     .05       0
  4958.5     .07       0  5004.9     .05       0
#XS Ineff= 2 , 0
         4745.74 1447.24    5250         1447.43
Permanent Ineff=
       F       F
Bank Sta=4958.5,4962.5
XS Rating Curve= 0 ,0
Exp/Cntr=0.3,0.1

Type RM Length L Ch R = 1 ,32500   ,500,500,500
BEGIN DESCRIPTION:
SAND SPRING CREEK 64.0
END DESCRIPTION:
XS GIS Cut Line= 3
      2771955.72     10289053.09      2770994.25     10289611.38
      2770805.69     10290903.08
#Sta/Elev= 30
  3888.2 1470.26  4122.6 1457.33  4276.1 1450.23  4415.2 1446.52  4736.4 1441.16
  4898.7 1440.09  4918.6 1440.05  4996.8 1438.83  5112.9 1440.22  5165.8 1439.61
  5274.6 1439.78  5294.8 1439.54  5303.8 1438.28  5304.1 1437.78  5307.8 1438.28
  5335.3 1439.47  5440.7 1441.74  5456.5 1441.06  5466.6 1442.21  5557.6  1444.3
  5759.7 1447.65  5779.9 1447.18  5785.6 1448.32  5891.1 1453.73  6083.1 1457.28
  6123.5 1460.17  6143.7 1459.74  6200.4 1462.81  6275.5 1463.83  6305.4 1465.42
#Mann= 6 ,-1 , 0
  3888.2     .12       0  4122.6     .05       0  4898.7     .12       0
  4918.6     .05       0  5165.8     .07       0  5335.3     .05       0
#XS Ineff= 2 , 0
         5115.91 1440.38
Permanent Ineff=
       F       F
Bank Sta=5303.8,5307.8
XS Rating Curve= 0 ,0
Exp/Cntr=0.3,0.1

Type RM Length L Ch R = 1 ,32000   ,500,500,500
BEGIN DESCRIPTION:
SAND SPRING CREEK 63.0
END DESCRIPTION:
XS GIS Cut Line= 3
      2771105.67     10288503.15      2770758.99     10289180.48
      2769955.68     10291103.11
#Sta/Elev= 30
  4239.1 1458.87  4449.1 1451.63  4497.4 1450.92  4513.9 1449.02  4562.1 1448.54
  4580.5 1448.23    4767 1443.63    4969 1435.82  4974.6 1434.33  4991.2 1434.62
  4994.8  1433.7  4995.1  1433.2  4998.8  1433.7  5020.3 1435.63  5111.2 1437.75
    5516 1438.19    5522 1438.27  5838.5 1439.01  5902.4 1439.97  6294.9 1443.78
  6373.2 1444.81  6474.4 1446.28  6477.2 1446.11  6606.8 1448.82  6631.8  1450.3
  6650.2 1449.64  6932.6  1455.8  7040.6 1457.25  7062.1 1457.81  7083.7 1458.25
#Mann= 16 ,-1 , 0
  4239.1     .05       0  4449.1     .12       0  4562.1     .05       0
  4580.5     .07       0    5516     .05       0    5522     .12       0
  5838.5     .05       0  5902.4     .12       0  6294.9     .05       0
  6373.2     .12       0  6474.4     .05       0  6477.2     .12       0
  6606.8     .05       0  6932.6     .12       0  7040.6     .05       0
  7062.1     .12       0
#XS Ineff= 2 , 0
                          5119.6         1437.82
Permanent Ineff=
       F       F
Bank Sta=4994.8,4998.8
XS Rating Curve= 0 ,0
Exp/Cntr=0.3,0.1

Type RM Length L Ch R = 1 ,31500   ,500,500,500
BEGIN DESCRIPTION:
SAND SPRING CREEK 62.0
END DESCRIPTION:
XS GIS Cut Line= 3
      2770905.68     10288453.11      2770497.74     10288784.53
      2770005.69     10289203.11
#Sta/Elev= 30
  4474.4 1456.53  4580.7 1451.31  4630.3 1450.31  4644.6 1448.44    4659 1448.65
  4844.3 1441.33  4879.5 1439.46  4893.9 1438.04  4914.7 1437.56  4995.9  1429.8
  4996.2  1429.3    5000  1429.3  5000.3  1429.8    5029  1432.9  5042.5 1434.65
  5071.1 1436.56    5171 1437.04    5305 1439.45  5333.6 1441.17  5347.8 1440.86
  5362.1 1442.16  5411.5  1443.7  5433.5 1445.48  5454.4 1445.55  5525.8 1448.93
  5567.5 1450.06  5589.5 1450.32    5596  1449.8  5610.3 1450.57    5646 1450.63
#Mann= 3 ,-1 , 0
  4474.4     .05       0  4914.7     .07       0    5029     .05       0
#XS Ineff= 2 , 0
                         5155.68         1437.33
Permanent Ineff=
       F       F
Bank Sta=4995.9,5000.3
XS Rating Curve= 0 ,0
Exp/Cntr=0.3,0.1

Type RM Length L Ch R = 1 ,31000   ,500,500,500
BEGIN DESCRIPTION:
SAND SPRING CREEK 61.0
END DESCRIPTION:
XS GIS Cut Line= 3
      2770305.69     10287903.08      2770213.98      10288394.6
      2769955.67     10289053.15
#Sta/Elev= 30
    4500 1449.52  4531.5 1450.39    4595 1447.64  4622.1 1445.99  4815.4 1437.89
  4866.2 1436.33  4876.4 1436.81  4947.6  1430.7  4968.2 1428.17  5004.2 1426.05
  5004.5 1425.55  5008.6 1426.05  5011.8  1427.1  5030.6 1428.11  5036.2  1428.4
  5041.6 1429.81  5060.6 1431.18  5073.6 1433.34  5114.9 1433.58  5120.2 1434.37
  5150.1  1433.1  5228.7 1434.21  5234.7 1435.05  5266.9 1435.66    5283 1434.92
  5337.2  1437.2  5406.6 1437.35  5428.1 1438.83  5492.5 1439.73  5707.4 1447.24
#Mann= 5 ,-1 , 0
    4500     .05       0    4595     .12       0  4622.1     .05       0
  4947.6     .07       0  5030.6     .05       0
#XS Ineff= 2 , 0
                         5115.36         1434.48
Permanent Ineff=
       F       F
Bank Sta=5004.2,5008.6
XS Rating Curve= 0 ,0
Exp/Cntr=0.3,0.1

Type RM Length L Ch R = 1 ,30500   ,500,500,500
BEGIN DESCRIPTION:
SAND SPRING CREEK 60.0
END DESCRIPTION:
XS GIS Cut Line= 3
      2769905.68     10287803.11      2769790.14     10288163.75
      2769605.67     10288403.12
#Sta/Elev= 30
  4621.3 1445.16  4631.8 1443.66  4637.4 1441.52  4776.2 1433.15  4789.3 1431.36
  4798.1 1431.99  4835.4 1430.57  4841.8 1429.31  4852.3  1429.9  4862.3 1429.29
  4867.6 1427.79  4894.3 1427.76    4905 1425.75  4925.8  1425.2  4957.3 1419.97
  4969.3 1416.71  4993.9 1415.39  4994.2 1414.89  4998.4 1415.39  5010.5 1416.54
  5016.8 1419.85  5037.6 1427.07  5045.8 1426.46  5052.1 1428.43  5074.8 1429.46
  5087.6 1431.43  5201.6  1435.2  5224.3 1436.74  5251.7 1436.49  5302.2 1438.76
#Mann= 4 ,-1 , 0
  4621.3     .12       0  4776.2     .05       0  4993.9     .05       0
  4998.4     .05       0
Bank Sta=4993.9,4998.4
XS Rating Curve= 0 ,0
Exp/Cntr=0.3,0.1

Type RM Length L Ch R = 1 ,30000   ,500,500,500
BEGIN DESCRIPTION:
SAND SPRING CREEK 59.0
END DESCRIPTION:
XS GIS Cut Line= 3
      2769555.71     10287653.07      2769433.18     10287831.08
      2769355.68     10288503.12
#Sta/Elev= 30
  4783.9  1439.8    4787  1439.8  4791.4 1437.04  4806.3 1432.03  4842.1 1425.88
  4848.2 1425.23  4856.8 1426.08  4928.7 1421.65  4964.6 1417.43  4978.2 1413.35
  4989.3 1411.64  4989.6 1411.14  4993.8 1411.64  5003.5 1412.67  5019.5 1419.03
  5024.5 1420.04  5072.5  1422.9    5143 1423.31  5197.4 1425.81  5213.4 1427.62
  5314.1 1429.02  5344.3 1431.19  5434.9 1433.11  5475.2 1433.14  5535.6 1434.94
  5543.1 1434.79  5548.1 1433.12    5632 1435.41    5637 1434.29  5676.5  1434.6
#Mann= 3 ,-1 , 0
  4783.9     .05       0  4989.3     .05       0  4993.8     .05       0
Bank Sta=4989.3,4993.8
XS Rating Curve= 0 ,0
Exp/Cntr=0.3,0.1

Type RM Length L Ch R = 1 ,29500   ,500,500,500
BEGIN DESCRIPTION:
SAND SPRING CREEK 58.0
END DESCRIPTION:
XS GIS Cut Line= 3
      2769455.68     10287453.11      2769062.83     10287527.32
      2768955.68     10288153.11
#Sta/Elev= 30
  4600.2 1434.08  4691.8 1427.43    4750 1424.58  4783.4 1423.12  4803.7 1420.92
  4813.4 1421.15  4824.1 1421.47  4864.8 1419.34  4885.1 1419.06  4956.4  1415.5
  4966.6 1414.25  4976.7 1411.86  4986.9 1409.38    4996 1406.04  5003.5 1405.59
  5003.8 1405.09  5007.9 1405.09  5008.3 1405.59  5011.8 1405.73  5016.9 1407.98
  5036.3 1411.56  5046.5 1414.27    5077 1417.78  5147.9  1418.6  5168.2 1419.63
  5178.3 1419.32  5427.2 1425.16  5432.3 1426.22  5462.4 1425.47  5634.9 1429.51
#Mann= 5 ,-1 , 0
  4600.2     .05       0    4750     .12       0  4813.4     .05       0
  5003.5     .05       0  5008.3     .05       0
Bank Sta=5003.5,5008.3
XS Rating Curve= 0 ,0
Exp/Cntr=0.3,0.1

Type RM Length L Ch R = 1 ,29000   ,500,500,500
BEGIN DESCRIPTION:
SAND SPRING CREEK 57.0
END DESCRIPTION:
XS GIS Cut Line= 3
      2769355.65     10287303.09      2768931.31     10287073.44
      2768455.66      10286853.1
#Sta/Elev= 30
  4517.5 1426.56  4607.4 1424.69  4738.6 1418.94  4799.5 1415.16  4824.2 1414.24
  4907.9 1410.56  4929.8 1411.16  4973.6 1406.15  4983.7  1404.5  4989.8 1402.27
  5003.8 1401.67  5004.1 1401.17  5008.6 1401.67  5012.2 1403.56  5035.1 1404.25
  5063.5 1408.36  5080.9 1409.56  5086.5 1408.83  5103.9 1410.97  5109.4 1410.44
  5126.8 1412.71  5160.7 1414.25  5178.1 1416.47  5206.5 1417.17  5269.8 1420.95
  5298.2 1421.46    5367 1425.37  5395.4 1425.72  5480.1 1429.24  5524.2 1432.16
#Mann= 5 ,-1 , 0
  4517.5     .05       0  4799.5     .12       0  4824.2     .05       0
  5003.8     .05       0  5008.6     .05       0
Bank Sta=5003.8,5008.6
XS Rating Curve= 0 ,0
Exp/Cntr=0.3,0.1

Type RM Length L Ch R = 1 ,28500   ,500,500,500
BEGIN DESCRIPTION:
SAND SPRING CREEK 56.0
END DESCRIPTION:
XS GIS Cut Line= 3
      2769505.69     10286703.11      2769104.77     10286610.84
      2768755.66     10286703.12
#Sta/Elev= 30
  4588.6 1422.47  4598.9 1422.44  4626.5 1419.86  4695.4 1415.91    4763 1412.09
  4804.1 1410.73  4827.2 1408.82  4879.7 1407.01  4886.2 1405.16    4917 1405.42
    4958 1402.53  4970.5 1401.42  4988.8 1396.17  4994.5 1395.72  4994.9 1395.22
  4999.4 1395.72  5026.7 1400.83  5031.8  1400.6  5061.1 1405.03  5072.1 1405.28
  5081.8 1403.73  5092.1 1405.19  5132.2 1407.28  5174.9 1409.01  5182.5 1410.63
  5195.6 1410.45    5263 1414.47  5288.7 1415.19    5330 1418.72  5361.1 1420.18
#Mann= 7 ,-1 , 0
  4588.6     .05       0  4626.5     .12       0  4695.4     .05       0
  4827.2     .12       0  4994.5     .07       0  4999.4     .12       0
  5132.2     .05       0
Bank Sta=4994.5,4999.4
XS Rating Curve= 0 ,0
Exp/Cntr=0.3,0.1

Type RM Length L Ch R = 1 ,28000   ,500,500,500
BEGIN DESCRIPTION:
SAND SPRING CREEK 55.0
END DESCRIPTION:
XS GIS Cut Line= 3
      2769555.68     10286403.11       2769156.5       10286140.
      2768655.69      10286553.1
#Sta/Elev= 30
  4521.9 1420.93  4571.6 1419.49  4608.4 1416.85    4674 1411.81  4736.2 1408.91
  4746.3 1407.89  4767.3  1407.9  4803.5 1404.01  4869.2 1402.59  4875.7 1401.35
  4881.7 1401.89  4890.8 1400.55  4896.8 1400.91  4911.9 1398.84  4932.9 1399.03
    4948 1396.04  4953.4 1396.94  4963.1  1394.6  4969.1 1395.58  4981.7 1392.53
    4982 1392.03  4986.6 1392.53  4997.5 1393.81  5016.6 1393.76    5031 1395.61
  5066.1 1397.84  5244.7 1403.46  5332.3 1407.65  5449.7 1412.81  5649.2 1422.98
#Mann= 9 ,-1 , 0
  4521.9     .05       0  4608.4     .12       0  4736.2     .05       0
  4953.4     .12       0  4981.7     .07       0  4986.6     .12       0
  5016.6     .05       0  5332.3     .12       0  5449.7     .05       0
Bank Sta=4981.7,4986.6
XS Rating Curve= 0 ,0
Exp/Cntr=0.3,0.1

Type RM Length L Ch R = 1 ,27500   ,500,500,500
BEGIN DESCRIPTION:
SAND SPRING CREEK 54.0
END DESCRIPTION:
XS GIS Cut Line= 3
      2769055.72      10285753.1      2768806.58     10285809.33
      2768605.68     10286053.12
#Sta/Elev= 30
  4744.6 1405.54    4786  1403.2    4812 1400.31  4817.1 1400.91  4826.6 1400.36
  4877.9 1396.34  4888.2 1396.04  4903.6 1394.15  4929.2 1393.47  4951.9 1391.61
  4970.2 1387.36  4990.5 1385.26  4995.4 1384.43  4995.8 1383.93    5000 1383.93
  5000.4 1384.43  5004.6 1384.43  5010.3 1386.78  5024.7 1388.55  5031.1  1392.6
  5045.5 1394.71  5053.3 1394.89  5059.8 1396.39  5074.2 1396.22  5160.2  1400.9
  5173.4 1400.43  5195.4 1402.01  5209.7 1401.79  5216.2 1402.48  5315.9 1405.85
#Mann= 5 ,-1 , 0
  4744.6     .05       0    4786     .12       0  4990.5     .05       0
  4995.4     .05       0  5000.4     .05       0
Bank Sta=4995.4,5000.4
XS Rating Curve= 0 ,0
Exp/Cntr=0.3,0.1

Type RM Length L Ch R = 1 ,27000   ,480,480,480
BEGIN DESCRIPTION:
SAND SPRING CREEK 53.0
END DESCRIPTION:
XS GIS Cut Line= 3
      2769205.71     10285753.15      2768965.27     10285346.98
      2768105.64     10285553.12
#Sta/Elev= 30
    4528 1403.16  4572.9 1402.58  4578.7 1403.19  4711.4 1397.79  4717.2 1398.19
  4797.1 1393.78    4865 1388.38  4923.1 1385.54  4951.2 1382.91  4966.8  1382.8
  4972.6 1381.26  4988.2 1382.47  5007.4 1381.18  5007.8 1380.68  5012.4 1381.18
  5020.1 1382.81  5046.8 1384.86  5081.8 1385.46  5112.7 1388.69  5130.8 1386.83
  5164.1 1386.41  5256.7 1386.94  5309.1 1389.36  5359.5 1389.91    5388 1392.08
    5472 1393.97  5734.4 1405.94    5812 1407.33  5842.8 1409.93    5884 1411.49
#Mann= 3 ,-1 , 0
    4528     .05       0  5007.4     .03       0  5012.4     .05       0
Bank Sta=5007.4,5012.4
XS Rating Curve= 0 ,0
Exp/Cntr=0.3,0.1

Type RM Length L Ch R = 1 ,26520   ,440,440,440
BEGIN DESCRIPTION:
Mapping XS 591e4f66
END DESCRIPTION:
XS GIS Cut Line= 3
      2769683.96     10285684.65      2769321.84     10285014.73
      2768271.71     10284743.15
#Sta/Elev= 30
  4292.9 1390.12  4316.3 1388.89  4343.8 1389.91  4381.9 1387.79  4616.9 1384.13
  4633.1 1382.84  4698.8 1381.59  4726.6 1382.38  4817.5 1379.33  4846.3 1379.09
  4911.9 1381.03    4950 1380.31  4965.3 1379.54  4991.3 1376.13  4991.6 1375.63
  4996.3 1376.13    5010 1376.76  5022.2 1379.38  5044.9  1380.3  5119.2 1380.46
  5174.4 1379.29  5184.7 1380.14    5226 1379.51  5267.4 1380.46  5649.5 1381.55
  5742.5 1382.62  5916.3 1386.76  5938.7 1385.89  6002.7 1387.06  6139.1 1386.25
#Mann= 3 ,-1 , 0
  4292.9     .05       0  4991.3     .05       0  4996.3     .05       0
Bank Sta=4991.3,4996.3
XS Rating Curve= 0 ,0
Exp/Cntr=0.3,0.1

Type RM Length L Ch R = 1 ,26080   ,580,580,580
BEGIN DESCRIPTION:
Mapping XS 5da30611
END DESCRIPTION:
XS GIS Cut Line= 3
      2770553.06      10286028.7      2770245.25     10285014.73
      2768670.33     10284580.28
#Sta/Elev= 30
  3408.5 1384.31  3466.6 1383.85  3516.8 1382.08    3522 1382.81  3549.7 1381.53
  3675.6 1380.73  3691.7 1381.44  3853.3 1378.08  3970.5    1377  4274.4 1368.87
  4274.8 1368.37  4279.4 1368.87  4302.6 1369.76  4459.4 1369.52  4924.1 1375.36
  4955.3  1375.3  4996.8 1371.52  5069.4 1376.85  5174.1 1375.01  5297.6 1374.88
  5411.7 1376.15  5629.5 1376.45  5650.3 1377.39  5696.7 1376.54  5816.3  1379.1
    5837 1378.11  5868.1 1379.27  5889.2 1378.12  6031.9 1377.77  6101.9 1379.84
#Mann= 3 ,-1 , 0
  3408.5     .05       0  4274.4     .05       0  4279.4     .05       0
Bank Sta=4274.4,4279.4
XS Rating Curve= 0 ,0
Exp/Cntr=0.3,0.1

Type RM Length L Ch R = 1 ,25500   ,500,500,500
BEGIN DESCRIPTION:
SAND SPRING CREEK 50.0
END DESCRIPTION:
XS GIS Cut Line= 3
      2771655.69     10285003.11      2769741.36     10284429.95
      2768980.66     10284428.11
#Sta/Elev= 30
  3001.7 1398.05  3194.1 1388.01  3260.3 1382.28  3331.7 1377.83  3481.9 1372.98
  3638.5 1373.74  3920.3 1369.31  3982.9 1370.12  4193.5  1368.6  4210.1 1368.11
  4210.4 1367.61  4215.1 1368.11  4382.5 1369.15  4552.5 1370.71  4772.3 1371.04
  4838.9 1372.36  4859.8 1371.76    4866 1372.57  4899.1 1371.24  4904.3 1372.09
  4943.3 1369.76  4975.9 1370.29    5000 1368.28  5025.7 1371.26  5055.7 1371.85
  5095.7 1370.54  5215.7  1370.6  5335.7 1372.21  5575.7 1373.36  5760.7 1376.71
#Mann= 7 ,-1 , 0
  3001.7     .05       0  4193.5     .12       0  4210.1     .05       0
  4215.1     .12       0  4382.5     .05       0  4772.3     .12       0
  4975.9     .05       0
Bank Sta=4210.1,4215.1
XS Rating Curve= 0 ,0
Exp/Cntr=0.3,0.1

Type RM Length L Ch R = 1 ,25000   ,1000,1000,1000
BEGIN DESCRIPTION:
SAND SPRING CREEK 49.0
END DESCRIPTION:
XS GIS Cut Line= 3
      2771655.72     10284953.13      2769758.75     10283958.95
      2769230.71     10283878.11
#Sta/Elev= 30
  2858.3 1396.89  2971.2 1391.29  3072.9 1384.04  3169.8 1378.27  3318.5 1373.89
  3456.7 1371.27  3748.5 1369.66  3842.4  1367.7  3989.4  1368.4  4098.4 1368.23
  4258.3 1366.74    4614 1367.62  4718.7 1367.13  4746.4 1365.82  4812.6 1365.38
  4917.2 1365.28  4939.3 1366.19  4969.6 1365.36  4983.4 1364.12  4992.2 1361.79
  4996.4 1361.67  4996.8 1361.17  5001.5 1361.67  5033.5 1362.89  5070.2 1366.14
    5165 1365.71  5185.2  1366.8  5367.3 1367.57  5438.1 1369.24  5534.2 1369.31
#Mann= 5 ,-1 , 0
  2858.3     .05       0  3989.4     .12       0  4098.4     .05       0
  4996.4     .05       0  5001.5     .05       0
Bank Sta=4996.4,5001.5
XS Rating Curve= 0 ,0
Exp/Cntr=0.3,0.1

Type RM Length L Ch R = 1 ,24000   ,500,500,500
BEGIN DESCRIPTION:
SAND SPRING CREEK 47.0
END DESCRIPTION:
XS GIS Cut Line= 3
      2772005.72     10285103.15      2770106.47     10283213.59
      2769105.68     10282803.11
#Sta/Elev= 30
  2320.9  1420.2    2328 1418.39  2349.2  1417.3  2356.3 1415.38  2405.8 1414.13
  2441.2 1409.33  2462.4 1408.85  2483.6 1411.25  2511.9 1407.11  2582.6 1402.66
    2625  1401.5  2999.8 1381.79    3120 1376.67  3339.2 1372.44  3452.3 1368.18
  3643.3 1364.56    3721 1365.12  3763.4 1362.91  3784.7 1364.02  4371.6 1367.55
  4866.5 1360.97  4993.7  1354.9  4994.2  1354.4  5000.4  1354.9  5015.7 1356.42
  5069.1 1355.98  5175.9 1360.18  5354.6 1363.63  5638.5 1366.52  6081.7 1375.87
#Mann= 3 ,-1 , 0
  2320.9     .05       0  4993.7     .03       0  5000.4     .05       0
Bank Sta=4993.7,5000.4
XS Rating Curve= 0 ,0
Exp/Cntr=0.3,0.1

Type RM Length L Ch R = 1 ,23500   ,500,500,500
BEGIN DESCRIPTION:
SAND SPRING CREEK 46.0
END DESCRIPTION:
XS GIS Cut Line= 3
      2772205.71     10284703.14      2770320.15     10282803.72
      2769305.73     10282703.12
#Sta/Elev= 30
  2323.6 1412.35  2500.4 1399.34  2641.8 1390.66  2677.2 1390.12  2726.7 1387.14
  2838.1 1382.67  2851.7 1382.11  2995.4 1375.46  3080.3 1372.71  3490.4 1363.17
  3582.3 1361.87  3603.5 1360.26  3610.6 1361.05  3900.5 1360.99    4049 1362.82
  4218.7 1363.04  4466.2 1361.59    4841 1357.79  4982.4 1353.07  4993.1 1350.89
  4993.6 1350.39  4999.9 1350.89  5044.7 1354.86  5145.2 1359.45  5446.7 1362.14
  5486.8 1363.81  5506.9 1363.24    5527 1364.66  5677.8 1365.49  6019.4 1373.35
#Mann= 5 ,-1 , 0
  2323.6     .05       0  2838.1     .12       0  2851.7     .05       0
  4993.1     .05       0  4999.9     .05       0
Bank Sta=4993.1,4999.9
XS Rating Curve= 0 ,0
Exp/Cntr=0.3,0.1

Type RM Length L Ch R = 1 ,23000   ,500,500,500
BEGIN DESCRIPTION:
SAND SPRING CREEK 45.0
END DESCRIPTION:
XS GIS Cut Line= 3
      2772455.69     10284253.12      2770563.54     10282369.19
      2769555.71     10282403.11
#Sta/Elev= 30
  2329.9 1398.36    2344 1399.12  2358.2 1396.69  2414.7 1393.58  2450.1 1393.22
  2469.7 1390.65  2598.6 1382.81  2803.7 1373.67  2980.4 1367.45  3220.9  1361.9
  3539.1 1358.97  3673.4 1355.63  3722.9 1357.25    4034 1359.36  4415.9 1358.11
  4606.8 1359.68    4826 1356.99  4960.4 1350.83  4988.6 1347.68  4991.6 1346.02
  4992.1 1345.52  4998.4 1346.02  5027.9 1349.16  5117.9 1352.33    5218 1358.26
  5688.2 1364.46  5718.3 1366.38  5768.3 1367.03  5798.3  1366.2  6008.4 1368.51
#Mann= 4 ,-1 , 0
  2329.9     .12       0  2469.7     .05       0  4991.6     .03       0
  4998.4     .05       0
Bank Sta=4991.6,4998.4
XS Rating Curve= 0 ,0
Exp/Cntr=0.3,0.1

Type RM Length L Ch R = 1 ,22500   ,500,500,500
BEGIN DESCRIPTION:
SAND SPRING CREEK 44.0
END DESCRIPTION:
XS GIS Cut Line= 3
      2772555.67      10283853.1      2770805.57     10281934.23
      2770105.65     10282003.11
#Sta/Elev= 30
  2402.9 1385.27  2459.3 1384.72  2579.6 1376.83  2735.6 1370.23  2955.2 1363.71
  3202.5 1360.52  3393.7 1354.42  3528.2 1353.16  3761.9 1355.28  4158.5 1355.86
  4250.4 1356.83  4342.3 1360.84  4349.7 1359.63  4363.9 1359.58  4434.2 1360.77
  4618.6  1358.2  4788.2 1353.84  4816.6 1354.17    4951 1345.86  4979.4 1344.96
  4993.6 1343.32  4993.9  1342.5  4994.4    1342  5000.8  1342.5  5037.3 1344.69
  5150.6 1348.21  5190.8  1351.6  5210.9 1352.27  5411.9 1355.62  5703.3 1364.49
#Mann= 3 ,-1 , 0
  2402.9     .05       0  4993.9     .03       0  5000.8     .05       0
Bank Sta=4993.9,5000.8
XS Rating Curve= 0 ,0
Exp/Cntr=0.3,0.1

Type RM Length L Ch R = 1 ,22000   ,500,500,500
BEGIN DESCRIPTION:
SAND SPRING CREEK 43.0
END DESCRIPTION:
XS GIS Cut Line= 3
      2771255.67     10281903.09      2771026.44     10281498.87
      2770505.65     10281453.11
#Sta/Elev= 30
  4535.3 1356.87  4564.9  1356.8  4753.8 1348.53  4844.7 1346.68  4882.8 1344.26
  4915.4 1342.39  4925.5  1342.9  4947.1 1340.45  4952.9  1339.1  4968.8 1338.35
  4974.5 1336.81  5002.9 1335.27  5008.8 1333.88  5009.3 1333.38  5015.7 1333.88
  5020.8 1334.78  5030.9 1338.32  5040.9 1340.22    5051  1339.6  5111.2 1341.16
  5231.6 1347.65  5236.9 1348.44  5245.2 1348.14  5281.8 1350.05  5291.9 1349.49
    5332 1351.92  5392.3 1353.86  5466.6 1355.35  5492.6 1356.73  5522.8 1356.57
#Mann= 5 ,-1 , 0
  4535.3     .05       0  4882.8     .12       0  5008.8     .07       0
  5015.7     .12       0  5245.2     .05       0
Bank Sta=5008.8,5015.7
XS Rating Curve= 0 ,0
Exp/Cntr=0.3,0.1

Type RM Length L Ch R = 1 ,21500   ,394,394,394
BEGIN DESCRIPTION:
SAND SPRING CREEK 42.0
END DESCRIPTION:
XS GIS Cut Line= 3
      2771405.69     10281553.14      2771304.54     10281131.09
      2770455.72     10281053.11
#Sta/Elev= 30
    4566 1348.28  4607.2 1346.93    4638 1348.32  4668.5 1345.29    4823 1339.25
  4905.4 1336.59  4925.8 1337.29  4936.2 1333.47  4967.7 1327.52  4972.9 1325.31
  4992.9 1322.32  4993.4 1321.82  4999.9 1322.32  5008.9 1322.51  5033.3 1327.42
  5143.2 1331.99  5229.8 1337.43  5290.1 1337.25  5300.1 1338.63  5357.9 1340.17
  5541.1 1341.94  5577.7 1340.61  5582.7 1337.85  5601.4 1341.29  5687.6 1346.87
  5692.6 1345.94  5772.1 1347.12  5792.2  1349.2  5812.3 1348.74  5852.4 1350.28
#Mann= 5 ,-1 , 0
    4566     .05       0    4823     .12       0  4967.7     .05       0
  4992.9     .03       0  4999.9     .05       0
Bank Sta=4992.9,4999.9
XS Rating Curve= 0 ,0
Exp/Cntr=0.3,0.1

Type RM Length L Ch R = 1 ,21106   ,444,444,444
BEGIN DESCRIPTION:
Mapping XS b8a79aa6
END DESCRIPTION:
XS GIS Cut Line= 3
      2771948.73      10281468.5      2771514.68     10280806.57
      2770744.25     10280632.96
#Sta/Elev= 30
  4306.5 1342.64    4326 1342.96  4348.8 1344.72  4356.2 1343.71  4377.3 1343.39
  4398.4 1344.34  4407.5    1343  4413.5 1343.66  4428.6 1340.22  4434.6 1340.65
  4443.7  1339.3  4528.2 1334.58  4543.1  1334.8  4552.1 1333.73  4723.9 1326.91
  4891.1 1323.87  4925.5 1322.63    4947 1322.68  4983.1 1320.91  4994.7 1318.32
  4995.2 1317.82  5001.7 1318.32  5006.5 1321.29  5013.3 1322.35  5127.8  1325.3
  5183.1 1324.47  5361.2 1325.14  5501.2 1324.57  5619.8 1326.02  5887.8 1326.13
#Mann= 5 ,-1 , 0
  4306.5     .05       0  4891.1     .12       0  4925.5     .05       0
  4994.7     .03       0  5001.7     .05       0
Bank Sta=4994.7,5001.7
XS Rating Curve= 0 ,0
Exp/Cntr=0.3,0.1

Type RM Length L Ch R = 1 ,20662   ,338,338,338
BEGIN DESCRIPTION:
Mapping XS ac7695dd
END DESCRIPTION:
XS GIS Cut Line= 3
      2772361.07     10280947.66       2771840.2     10280589.56
      2770799.65     10280416.14
#Sta/Elev= 30
  4315.2 1322.44    4336 1321.84  4479.5 1321.97  4494.3 1321.42  4616.8  1320.8
  4754.1 1321.36  4775.1 1320.58  4831.9 1321.01  4927.3 1319.95  4933.4 1320.56
    4947 1319.56  4956.5 1319.84  4999.1 1315.44  4999.6 1314.94  5005.6 1314.94
  5006.1 1315.44  5012.3 1318.17  5017.4  1317.3  5022.8 1318.41  5144.5 1320.91
  5194.8 1321.29  5286.4 1321.65  5296.6 1321.08  5347.3 1321.68  5387.8 1321.19
  5428.4 1321.69  5651.4 1321.27  5702.1 1321.76  5813.6 1321.26  6002.2 1322.75
#Mann= 3 ,-1 , 0
  4315.2     .05       0  4999.1     .05       0  5006.1     .05       0
Bank Sta=4999.1,5006.1
XS Rating Curve= 0 ,0
Exp/Cntr=0.3,0.1

Type RM Length L Ch R = 1 ,20324   ,740,740,740
BEGIN DESCRIPTION:
Mapping XS ebe2b85b
END DESCRIPTION:
XS GIS Cut Line= 4
      2772447.88     10280567.88       2771883.6     10280274.89
      2771579.79     10280231.49      2770940.16     10280209.81
#Sta/Elev= 30
  4232.6 1318.07  4280.6 1317.19  4325.2 1318.24  4424.2 1317.97  4606.9 1316.43
  4728.2    1318  4800.2 1317.47  4896.6 1318.83    4937 1318.51  4957.2 1317.28
  4977.4 1315.87  4984.8 1313.69  4989.8 1314.37  4994.1 1312.88  4994.6 1312.38
  5001.1 1312.88  5017.8 1315.22    5038 1316.25  5131.2 1316.24  5169.3  1317.6
  5229.4 1318.06  5259.5 1319.57  5289.5 1319.13  5299.5 1320.04  5309.5 1319.38
  5329.5 1320.15  5419.5 1319.15  5449.6 1319.89  5719.7 1319.78  5815.3 1320.86
#Mann= 3 ,-1 , 0
  4232.6     .05       0  4994.1     .05       0  5001.1     .05       0
Bank Sta=4994.1,5001.1
XS Rating Curve= 0 ,0
Exp/Cntr=0.3,0.1

Type RM Length L Ch R = 1 ,19584   ,584,584,584
BEGIN DESCRIPTION:
Mapping XS 489732ee
END DESCRIPTION:
XS GIS Cut Line= 5
      2772556.35      10280426.8      2772219.98     10280122.98
      2771905.31     10279764.91      2771634.04      10279634.7
       2770993.8      10279634.7
#Sta/Elev= 30
  4232.8 1316.24  4257.3  1316.8  4441.1 1314.23  4469.5 1315.29  4547.3 1314.02
  4685.6 1315.35  4766.6 1315.45  4837.7 1314.17    4859 1314.76  4915.6 1313.42
  4929.8 1313.84  4979.1 1312.19  4986.7 1311.06  4989.9 1307.92  4990.4 1307.42
  4996.9 1307.92  5007.6 1310.48  5036.1 1311.68    5072 1311.53  5142.3 1312.96
  5184.5 1311.57  5217.8 1311.73    5224 1311.95  5229.6 1313.42  5246.7 1313.03
  5252.2 1314.85  5395.3 1316.69    5782 1318.59    5912 1317.52  6103.9 1319.61
#Mann= 3 ,-1 , 0
  4232.8     .05       0  4989.9     .05       0  4996.9     .05       0
Bank Sta=4989.9,4996.9
XS Rating Curve= 0 ,0
Exp/Cntr=0.3,0.1

Type RM Length L Ch R = 1 ,19000   ,500,500,500
BEGIN DESCRIPTION:
SAND SPRING CREEK 38.0
END DESCRIPTION:
XS GIS Cut Line= 3
       2772955.7     10281353.15      2772393.14     10279461.63
      2772155.68     10278453.11
#Sta/Elev= 30
  3026.6 1335.81  3362.8 1323.78  3462.4  1323.8  3475.3  1321.6  3500.8 1323.54
  4038.6 1313.98  4424.6 1309.87  4581.1    1311  4868.2 1306.44  4967.2 1307.12
  4996.6 1303.39  5054.7 1307.71  5193.7 1308.53  5361.5 1305.19  5374.9 1302.56
  5375.4 1302.06  5382.3 1302.56  5403.8 1306.27  5531.2 1310.73  5625.9  1315.6
  5645.7 1319.51  5668.3 1317.76  5717.6 1322.38  5738.2 1320.88  5758.7 1323.66
  5819.4 1325.26  5912.8 1329.43  5975.1  1324.7    5995 1333.38  6036.1 1336.77
#Mann= 5 ,-1 , 0
  3026.6     .05       0  5374.9     .05       0  5382.3     .05       0
  5531.2     .12       0  5819.4     .05       0
Bank Sta=5374.9,5382.3
XS Rating Curve= 0 ,0
Exp/Cntr=0.3,0.1

Type RM Length L Ch R = 1 ,18500   ,500,500,500
BEGIN DESCRIPTION:
SAND SPRING CREEK 37.0
END DESCRIPTION:
XS GIS Cut Line= 3
      2772855.68     10280153.07      2772733.69     10279163.86
      2772705.68     10278953.11
#Sta/Elev= 30
  4003.3 1313.72  4073.8 1311.54  4154.4 1311.17  4272.6 1308.67  4284.8 1307.77
  4295.5 1305.57  4335.8  1304.1  4365.9 1305.33  4386.1 1307.83  4406.3 1306.31
  4436.5 1306.11  4446.6 1304.44  4452.1 1300.76    4483 1304.61    4507 1305.43
  4577.6 1303.59    4628  1303.8  4776.7 1298.38  4809.3 1299.73  4889.9 1299.59
  4944.1 1297.55  4993.9  1292.7  4994.4  1292.2  5001.9  1292.7  5010.8 1292.82
  5019.4 1295.15  5081.5 1305.43  5102.7 1306.28  5131.9  1309.7  5212.6 1315.66
#Mann= 5 ,-1 , 0
  4003.3     .05       0  4272.6     .12       0    4483     .05       0
  4993.9     .05       0  5001.9     .05       0
Bank Sta=4993.9,5001.9
XS Rating Curve= 0 ,0
Exp/Cntr=0.3,0.1

Type RM Length L Ch R = 1 ,18000   ,500,500,500
BEGIN DESCRIPTION:
SAND SPRING CREEK 36.0
END DESCRIPTION:
XS GIS Cut Line= 3
       2774155.7     10279403.12      2773185.76     10279064.63
      2773005.68      10278853.1
#Sta/Elev= 30
  3972.7  1339.4  4019.3 1337.59  4045.1 1334.31  4050.4  1334.9  4076.1 1330.78
  4169.3 1320.85  4293.6 1309.29  4449.3 1300.85  4681.5 1291.13  4743.6 1287.23
  4767.1 1286.96  4798.8  1284.9  4805.7 1283.19  4830.6  1283.4  4847.3 1282.21
  4847.8 1281.71  4856.3 1282.21  4904.8 1284.78  4921.6 1284.19  4978.9 1284.33
  4986.8 1283.84  4992.1 1282.24  5008.2 1282.61  5022.5 1286.32    5029 1286.69
  5036.8 1289.44  5042.1  1288.7  5079.6 1293.86  5164.1 1301.53  5277.8 1309.17
#Mann= 5 ,-1 , 0
  3972.7     .05       0  4847.3     .07       0  4856.3     .05       0
  4921.6     .12       0  5042.1     .05       0
Bank Sta=4847.3,4856.3
XS Rating Curve= 0 ,0
Exp/Cntr=0.3,0.1

Type RM Length L Ch R = 1 ,17500   ,500,500,500
BEGIN DESCRIPTION:
SAND SPRING CREEK 35.0
END DESCRIPTION:
XS GIS Cut Line= 3
      2773955.64     10279003.09      2773569.56      10278772.3
       2773055.7     10278703.11
#Sta/Elev= 30
  4550.2 1314.98  4674.7 1301.71  4680.5 1301.55  4696.1 1299.37  4701.9 1299.31
    4733 1295.49  4791.4 1290.75  4828.3 1289.18  4841.4  1287.8  4849.7 1285.06
  4855.6 1286.48  4871.1 1281.94  4892.5 1281.54  4908.1 1283.01  4913.9 1280.66
  4945.1 1278.34  4950.9 1279.08  4993.9 1274.66  4994.4 1274.16  5004.3 1274.16
  5004.8 1274.66    5014  1276.3  5030.3    1277  5044.3 1276.67  5094.7 1278.28
  5103.1 1279.54  5155.3 1284.06    5236 1288.32  5316.7 1294.59  5518.5 1307.27
#Mann= 3 ,-1 , 0
  4550.2     .05       0  4993.9     .05       0  5004.8     .05       0
Bank Sta=4993.9,5004.8
XS Rating Curve= 0 ,0
Exp/Cntr=0.3,0.1

Type RM Length L Ch R = 1 ,17000   ,500,500,500
BEGIN DESCRIPTION:
SAND SPRING CREEK 34.0
END DESCRIPTION:
XS GIS Cut Line= 3
      2774055.68     10278253.11      2773664.62      10278284.2
      2773155.69     10278553.11
#Sta/Elev= 30
  4607.7 1292.68  4627.8 1292.12  4647.8  1292.7  4666.8 1290.96  4671.8 1291.81
  4677.9  1290.1  4738.1 1287.97  4908.6 1274.46  4958.8 1272.55  4978.9  1271.3
  4991.5 1269.45    4992 1268.95  5002.5 1269.45  5006.4  1270.5  5012.1 1270.22
  5028.4 1272.22  5034.1    1272  5072.4 1275.73  5116.5 1277.67  5132.8 1279.76
  5138.5 1279.56  5176.9 1282.78  5198.9    1283  5204.5 1281.47  5264.9 1284.22
  5281.3 1283.85  5286.9 1285.46  5292.9 1286.01    5463 1290.94  5575.6 1296.48
#Mann= 3 ,-1 , 0
  4607.7     .05       0  4991.5     .05       0  5002.5     .05       0
Bank Sta=4991.5,5002.5
XS Rating Curve= 0 ,0
Exp/Cntr=0.3,0.1

Type RM Length L Ch R = 1 ,16500   ,500,500,500
BEGIN DESCRIPTION:
SAND SPRING CREEK 33.0
END DESCRIPTION:
XS GIS Cut Line= 3
      2773955.69     10278203.12      2773682.78     10277802.43
      2773505.71     10277603.14
#Sta/Elev= 30
  4515.2 1289.44  4579.6 1287.98  4609.4 1286.18  4624.1 1286.13  4645.4 1284.06
  4681.3 1282.63  4687.3 1282.94  4708.8 1281.19  4732.1 1280.77  4738.2 1278.99
  4745.1 1279.71  4759.1 1278.42  4781.4 1277.58  4817.7 1273.83  4866.9 1270.47
  4968.6  1267.8    4975 1266.11  4983.5 1266.47    4991 1264.12  4991.5 1263.62
  5001.6 1263.62  5002.1 1264.12    5012 1266.21  5018.7 1266.24  5025.8 1267.25
  5047.1 1271.59  5146.2 1282.91  5153.3 1282.72  5188.4 1285.71  5266.6 1289.99
#Mann= 3 ,-1 , 0
  4515.2     .05       0    4991     .05       0  5002.1     .05       0
Bank Sta=4991,5002.1
XS Rating Curve= 0 ,0
Exp/Cntr=0.3,0.1
