HEC-RAS study SIXMILE CREEK.prj: SIXMILE CREEK Base Level Engineering

--- SIXMILE CREEK.g01 (geometry) --- (continued)

Type RM Length L Ch R = 1 ,44500   ,500,500,500
BEGIN DESCRIPTION:
SIXMILE CREEK 89.0
END DESCRIPTION:
XS GIS Cut Line= 3
      2785755.68     10207403.11      2786122.56     10207327.94
       2786355.7     10207103.09
#Sta/Elev= 30
  4625.5 1302.62  4635.7 1300.94  4650.7 1299.86  4666.3 1295.59    4696 1289.44
  4701.1 1289.06  4746.5 1276.42  4751.6 1276.07  4758.2 1273.34  4778.6 1269.97
    4802 1264.26  4809.2  1261.2  4824.9 1257.38  4852.4 1250.39  4880.7 1245.14
  4902.9 1242.21  4926.6 1240.93  4931.7 1240.75  4939.7 1236.97  4940.2 1236.47
  4956.2 1236.47  4956.7 1236.97  4972.6 1237.87  5001.1 1237.18  5033.1 1238.93
  5083.5 1244.57  5132.9 1248.15  5210.8 1253.18  5260.2 1255.23  5323.9  1258.6
#Mann= 8 ,-1 , 0
  4625.5     .12       0  4824.9     .05       0  4926.6     .12       0
  4939.7     .07       0  4956.7     .12       0  5001.1     .05       0
  5033.1     .12       0  5260.2     .05       0
Bank Sta=4939.7,4956.7
XS Rating Curve= 0 ,0
Exp/Cntr=0.3,0.1

Type RM Length L Ch R = 1 ,44000   ,500,500,500
BEGIN DESCRIPTION:
SIXMILE CREEK 88.0
END DESCRIPTION:
XS GIS Cut Line= 3
      2786005.69     10207903.11      2786492.91     10207662.94
      2786755.71     10207453.09
#Sta/Elev= 30
  4456.8 1278.15  4493.3 1275.45  4501.4 1273.92  4577.5 1266.39    4600 1265.28
    4628 1262.48  4650.5 1261.81  4657.5 1259.89  4712.3 1255.59  4717.8 1254.28
  4734.7 1253.93    4769 1250.23  4802.1 1248.73  4835.9 1245.62  4869.3 1244.99
  4936.2 1238.31    4948 1234.07  4956.4 1233.83  4956.9 1233.33  4973.4 1233.83
  5052.1 1237.31  5072.9 1240.39  5087.3 1241.34  5093.7 1242.86    5201 1249.08
  5229.8 1249.85  5250.6 1252.63  5272.3 1253.46  5314.7 1257.81  5336.3    1259
#Mann= 3 ,-1 , 0
  4456.8     .05       0  4956.4     .03       0  4973.4     .05       0
Bank Sta=4956.4,4973.4
XS Rating Curve= 0 ,0
Exp/Cntr=0.3,0.1

Type RM Length L Ch R = 1 ,43500   ,500,500,500
BEGIN DESCRIPTION:
SIXMILE CREEK 87.0
END DESCRIPTION:
XS GIS Cut Line= 3
       2786505.7     10208103.11      2786849.91     10208009.93
      2787105.67     10207953.11
#Sta/Elev= 30
  4643.4 1253.52  4665.9  1251.7  4757.3 1247.31  4775.1 1245.64  4780.3 1246.32
  4840.2 1241.57  4849.6  1241.6  4854.8 1240.73  4881.7 1241.61  4889.5 1240.93
  4894.7 1239.58  4934.5 1235.58    4964  1233.8    5000 1233.39  5001.2 1232.86
  5001.7 1232.36  5017.7 1232.36  5018.2 1232.86  5026.4 1232.93  5046.9 1235.02
  5058.4 1237.62  5067.4 1238.62  5096.8 1239.63  5108.4 1241.66  5128.8 1242.59
  5145.5 1244.33  5169.8 1245.79  5200.5 1249.73  5237.7 1253.44    5262 1254.85
#Mann= 3 ,-1 , 0
  4643.4     .05       0  5001.2     .03       0  5018.2     .05       0
Bank Sta=5001.2,5018.2
XS Rating Curve= 0 ,0
Exp/Cntr=0.3,0.1

Type RM Length L Ch R = 1 ,43000   ,500,500,500
BEGIN DESCRIPTION:
SIXMILE CREEK 86.0
END DESCRIPTION:
XS GIS Cut Line= 3
      2786505.73      10208553.1      2787025.55     10208471.41
      2787405.69      10208103.1
#Sta/Elev= 30
  4473.8 1253.72  4575.2 1248.67  4595.2 1246.53  4632.7 1246.93  4676.2 1245.62
  4706.6  1243.5  4747.1 1243.03  4797.7 1240.41  4848.3 1239.38  4939.4 1232.66
  4947.2 1230.15  4947.7 1229.65  4964.3 1230.15  4997.5 1232.53  5027.3 1231.79
  5034.2 1230.51  5062.5 1230.78  5069.7 1233.11  5111.9 1235.72  5119.1 1237.85
  5154.4 1237.79  5161.6 1239.42  5168.5 1238.16  5175.7  1239.5  5218.2  1241.2
  5239.3 1243.76  5281.7 1245.97  5324.2 1250.61    5409 1256.56  5529.3 1262.05
#Mann= 3 ,-1 , 0
  4473.8     .05       0  4947.2     .05       0  4964.3     .05       0
Bank Sta=4947.2,4964.3
XS Rating Curve= 0 ,0
Exp/Cntr=0.3,0.1

Type RM Length L Ch R = 1 ,42500   ,500,500,500
BEGIN DESCRIPTION:
SIXMILE CREEK 85.0
END DESCRIPTION:
XS GIS Cut Line= 3
       2786155.7     10208403.12      2787157.18      10208950.7
      2787555.73     10209053.12
#Sta/Elev= 30
  3858.6 1271.08  3932.1 1267.69  3961.2 1263.13  4006.7 1260.42  4019.4  1261.2
  4035.5 1258.41  4079.1 1258.69  4132.1 1254.91  4204.4 1255.19  4302.1  1251.6
  4411.2 1249.96  4574.3 1242.98  4861.5 1234.61  4890.2 1230.69  5010.6 1226.68
  5011.1 1226.18  5027.7 1226.68  5039.8 1229.49  5108.5 1236.42  5230.7 1241.54
  5246.3 1243.81  5271.5 1244.36    5307 1249.94  5311.4  1248.6  5347.8 1255.24
  5352.9 1253.64  5370.2 1258.07  5388.5 1258.43  5393.7 1256.46  5411.5 1257.63
#Mann= 4 ,-1 , 0
  3858.6     .05       0  5010.6     .03       0  5027.7     .05       0
  5311.4     .12       0
Bank Sta=5010.6,5027.7
XS Rating Curve= 0 ,0
Exp/Cntr=0.3,0.1

Type RM Length L Ch R = 1 ,42000   ,500,500,500
BEGIN DESCRIPTION:
SIXMILE CREEK 84.0
END DESCRIPTION:
XS GIS Cut Line= 3
      2786155.67      10208453.1      2787169.11     10209446.18
      2788105.72     10209653.12
#Sta/Elev= 30
  3581.1 1269.28  3588.2 1269.72  3673.1 1262.97  3814.5 1256.49  3998.4 1251.26
  4111.5  1249.5  4203.4 1245.44  4373.1 1241.56  4528.7 1240.13  4641.9 1237.08
    4861 1235.98  4953.1 1225.08    5018 1223.63  5018.5 1223.13  5036.4 1223.63
  5059.2 1226.16  5097.7 1226.62  5102.8 1228.86  5139.9 1233.99  5146.5 1232.85
  5151.6 1236.58  5190.2 1236.45    5232 1231.51  5303.7  1237.7  5428.9 1240.44
  5733.9 1254.24  5891.1 1268.39    5908  1271.4  5934.8 1273.74  5959.2  1274.1
#Mann= 3 ,-1 , 0
  3581.1     .05       0    5018     .03       0  5036.4     .05       0
Bank Sta=5018,5036.4
XS Rating Curve= 0 ,0
Exp/Cntr=0.3,0.1

Type RM Length L Ch R = 1 ,41500   ,500,500,500
BEGIN DESCRIPTION:
SIXMILE CREEK 83.0
END DESCRIPTION:
XS GIS Cut Line= 3
      2786405.65     10209353.08      2786921.75     10209854.41
      2787005.69     10210103.12
#Sta/Elev= 30
  4280.5  1241.6  4464.3 1234.59  4563.4  1232.7  4605.8 1230.45  4641.3 1231.43
  4676.5 1227.91  4690.7 1228.21    4712 1231.27  4754.5 1233.76    4818 1234.33
  4874.6 1231.43  4881.6 1229.72    4924 1224.37  4945.8 1223.96  4980.6 1221.93
  4987.8  1222.4  4999.9  1220.7  5000.4  1220.2  5018.4  1220.7  5020.6 1221.43
  5031.8 1221.76  5040.8 1224.04  5051.4 1229.28    5058 1235.59  5072.5 1239.03
  5120.9 1240.67  5146.4 1239.92  5246.8 1248.56    5252  1247.9  5262.5 1249.06
#Mann= 5 ,-1 , 0
  4280.5     .05       0  4945.8     .12       0  4999.9     .07       0
  5018.4     .12       0  5020.6     .05       0
Bank Sta=4999.9,5018.4
XS Rating Curve= 0 ,0
Exp/Cntr=0.3,0.1

Type RM Length L Ch R = 1 ,41000   ,598,598,598
BEGIN DESCRIPTION:
SIXMILE CREEK 82.0
END DESCRIPTION:
XS GIS Cut Line= 3
      2786355.68     10209303.09      2786428.47     10209796.55
      2786505.68     10210053.08
#Sta/Elev= 30
  4501.2 1243.94    4536 1242.54    4572 1239.69  4670.3 1235.63  4753.9 1232.52
  4834.8 1230.95  4874.2 1227.66  4879.2 1229.93  4935.9 1223.18  5004.8 1220.91
  5028.4 1220.73  5028.9 1220.23  5046.4 1220.23  5046.9 1220.73  5048.6  1221.8
  5069.5 1221.05  5075.9 1222.63  5081.1 1222.51  5100.8 1224.23  5114.1 1224.27
  5141.9 1226.25  5147.2 1226.12  5153.1  1227.1  5173.9 1228.77  5194.8 1232.99
  5208.5 1234.63  5226.2 1238.38  5246.2 1241.29  5257.5 1244.29  5267.9 1244.71
#Mann= 5 ,-1 , 0
  4501.2     .05       0  5004.8     .12       0  5028.4     .03       0
  5046.9     .12       0  5208.5     .05       0
Bank Sta=5028.4,5046.9
XS Rating Curve= 0 ,0
Exp/Cntr=0.3,0.1

Type RM Length L Ch R = 1 ,40402   ,402,402,402
BEGIN DESCRIPTION:
SIXMILE CREEK 81.0
END DESCRIPTION:
XS GIS Cut Line= 3
      2785780.69     10209478.14      2785807.48     10209826.46
      2786380.72     10210078.13
#Sta/Elev= 30
  4566.3 1242.57  4741.8 1236.22  4872.2 1229.57  4935.5 1228.51  4948.3  1219.3
  4956.9 1216.65  4957.4 1216.15  4975.4 1216.65  4989.5 1219.41  5001.1 1217.09
  5047.2 1220.82  5099.4 1222.78    5164 1221.45  5169.4 1219.48  5192.8 1218.84
  5198.3 1221.89  5230.4  1223.8  5252.2  1223.5  5277.5 1226.02  5302.9 1227.43
  5343.9 1230.09  5361.5 1229.87  5367.2 1230.89  5372.7 1233.53  5383.3 1233.38
  5413.9 1237.37  5419.4  1236.5  5437.3 1238.92  5442.8 1237.78  5541.7    1242
#Mann= 5 ,-1 , 0
  4566.3     .05       0  4956.9     .03       0  4975.4     .05       0
  5277.5     .12       0  5302.9     .05       0
Bank Sta=4956.9,4975.4
XS Rating Curve= 0 ,0
Exp/Cntr=0.3,0.1

Type RM Length L Ch R = 1 ,40000   ,500,500,500
BEGIN DESCRIPTION:
SIXMILE CREEK 80.0
END DESCRIPTION:
XS GIS Cut Line= 3
      2784793.35     10210306.42      2785667.22     10210192.24
       2785905.7     10210303.12
#Sta/Elev= 30
  4118.7 1243.09  4201.8 1240.04  4337.5 1236.04  4411.4 1232.57  4520.5 1229.98
  4685.8 1227.06  4722.1 1224.73  4727.2 1225.61  4746.6 1225.09  4766.5 1224.98
  4786.7 1227.36  4816.9 1221.36    4827 1220.03  4847.2 1220.27  4874.9 1215.57
    4880 1216.72  4887.5 1215.76  4968.2 1215.93  4978.3 1214.65    5000 1215.56
    5021 1214.52  5021.5 1214.02  5041.7 1214.52  5053.4 1221.28  5060.2 1223.73
  5075.5  1226.1  5170.5 1230.78  5174.2 1230.75  5231.4 1235.18    5263 1235.73
#Mann= 8 ,-1 , 0
  4118.7     .12       0  4201.8     .05       0  4520.5     .12       0
  4746.6     .05       0    5021     .05       0  5041.7     .05       0
  5170.5     .12       0  5174.2     .05       0
Bank Sta=5021,5041.7
XS Rating Curve= 0 ,0
Exp/Cntr=0.3,0.1

Type RM Length L Ch R = 1 ,39500   ,500,500,500
BEGIN DESCRIPTION:
SIXMILE CREEK 79.0
END DESCRIPTION:
XS GIS Cut Line= 3
      2785255.69     10210753.11      2785478.41     10210636.49
       2785855.7      10210453.1
#Sta/Elev= 30
  4748.6 1240.43  4778.9    1237  4816.3 1234.71    4823 1233.16  4883.6 1229.28
  4895.3 1227.58  4933.3 1225.27  4949.8 1222.82  4955.4 1219.52  4963.1 1216.84
  4971.8 1212.23  4977.5 1210.51  4987.9 1209.97  4988.4 1209.47  5008.2 1209.47
  5008.7 1209.97    5022 1210.44  5039.1 1212.39  5052.6 1213.88  5067.1 1214.12
  5112.2 1216.76  5129.2 1222.33    5186 1226.94  5230.5 1229.23  5337.8 1232.28
  5365.9 1234.34  5382.9  1233.6  5388.4 1234.97  5404.4 1235.09  5419.5 1235.68
#Mann= 5 ,-1 , 0
  4748.6     .12       0  4987.9     .07       0  5008.7     .12       0
  5039.1     .05       0  5404.4     .12       0
Bank Sta=4987.9,5008.7
XS Rating Curve= 0 ,0
Exp/Cntr=0.3,0.1

Type RM Length L Ch R = 1 ,39000   ,500,500,500
BEGIN DESCRIPTION:
SIXMILE CREEK 78.0
END DESCRIPTION:
XS GIS Cut Line= 3
      2785805.69     10211103.08      2785876.88     10210856.97
      2786105.69      10210503.1
#Sta/Elev= 30
  4743.8 1229.31  4794.2 1227.97    4833 1225.72    4848 1224.31  4889.5 1221.21
  4899.9 1220.94    4939 1216.29  4965.2 1214.26  4972.6 1213.45  4977.8 1213.57
  4983.2  1212.2  4999.4 1210.05  5055.7 1208.63  5056.2 1208.13  5076.2 1208.13
  5076.7 1208.63  5096.5 1213.03  5117.6 1213.54  5132.8 1215.87  5138.7  1214.2
  5159.8 1216.21  5169.1 1218.19  5205.3 1220.62  5226.5 1223.41  5283.8 1225.49
    5299 1226.75  5320.1 1226.82  5326.1 1227.68  5344.7 1228.59  5421.4 1236.09
#Mann= 6 ,-1 , 0
  4743.8     .05       0    4848     .12       0  4965.2     .05       0
  5055.7     .05       0  5076.7     .05       0  5344.7     .12       0
Bank Sta=5055.7,5076.7
XS Rating Curve= 0 ,0
Exp/Cntr=0.3,0.1

Type RM Length L Ch R = 1 ,38500   ,500,500,500
BEGIN DESCRIPTION:
SIXMILE CREEK 77.0
END DESCRIPTION:
XS GIS Cut Line= 3
      2785955.66     10211703.16      2786366.97      10210774.9
      2786305.68     10210553.11
#Sta/Elev= 30
  3984.7 1255.29  4022.4 1257.01  4045.7    1254  4051.2 1254.66    4069 1251.58
  4074.4 1251.52  4083.2 1249.74  4115.5 1245.57  4225.4 1238.08    4440 1230.19
  4706.6 1222.55  4772.3 1221.56  4813.9 1219.25    4827 1218.61  4892.6 1218.34
  4961.7 1212.34    4969  1208.8  4969.5  1208.3    4990  1208.8  5074.1 1210.71
  5084.9  1213.9  5099.6 1214.58  5105.6 1218.37    5116 1220.54  5133.9 1222.27
  5139.1 1221.96  5167.9 1226.25  5173.4 1227.94  5227.8 1232.42  5230.1 1232.42
#Mann= 6 ,-1 , 0
  3984.7     .05       0  4813.9     .12       0    4969     .07       0
    4990     .12       0  5074.1     .05       0  5227.8     .12       0
Bank Sta=4969,4990
XS Rating Curve= 0 ,0
Exp/Cntr=0.3,0.1

Type RM Length L Ch R = 1 ,38000   ,500,500,500
BEGIN DESCRIPTION:
SIXMILE CREEK 76.0
END DESCRIPTION:
XS GIS Cut Line= 3
      2786605.71     10211303.07      2786818.82     10210905.71
      2786905.72     10210853.09
#Sta/Elev= 30
  4549.1 1226.47  4617.1 1223.88  4688.7 1218.35    4742 1216.92  4770.8 1217.33
  4798.7 1215.93    4809 1214.08  4814.6 1215.14  4821.4 1213.62  4830.9 1215.33
  4866.8  1214.4  4889.5  1212.8  4924.3 1208.39  4968.9 1207.67  4978.7 1206.71
  4981.1 1204.69  4981.6 1204.19  5002.1 1204.69    5008 1206.63  5014.3 1206.97
  5029.8 1209.89  5035.6 1213.03  5051.1 1218.19    5057 1221.76  5072.5 1226.01
  5078.3 1228.88    5088 1230.51  5095.6 1234.28  5098.6 1235.56  5101.6 1235.56
#Mann= 4 ,-1 , 0
  4549.1     .05       0  4981.1     .05       0  5002.1     .05       0
  5095.6     .12       0
Bank Sta=4981.1,5002.1
XS Rating Curve= 0 ,0
Exp/Cntr=0.3,0.1

Type RM Length L Ch R = 1 ,37500   ,500,500,500
BEGIN DESCRIPTION:
SIXMILE CREEK 75.0
END DESCRIPTION:
XS GIS Cut Line= 3
      2786805.73      10211353.1      2787176.76     10211254.14
      2787255.69      10210903.1
#Sta/Elev= 30
    4616 1224.66  4626.3 1224.82  4667.7 1222.11  4677.2 1220.65  4698.8 1219.77
  4713.6 1218.22  4729.8 1217.95  4753.7 1215.57  4802.2 1212.42  4822.9 1211.55
  4835.6 1211.93    4884 1211.15  4903.8 1210.84  4916.1 1207.79  4943.9 1207.26
  4967.8 1204.79  5000.8 1203.71  5001.3 1203.21  5021.8 1203.71  5022.3  1205.6
  5042.1 1208.13  5060.5 1213.02  5065.6 1217.04  5083.1 1216.51  5103.6 1219.46
    5114 1220.05  5157.3  1220.3    5165 1221.58    5206 1221.97  5359.8 1226.73
#Mann= 6 ,-1 , 0
    4616     .12       0  4677.2     .05       0  4835.6     .12       0
    4884     .05       0  5000.8     .03       0  5021.8     .05       0
Bank Sta=5000.8,5021.8
XS Rating Curve= 0 ,0
Exp/Cntr=0.3,0.1

Type RM Length L Ch R = 1 ,37000   ,500,500,500
BEGIN DESCRIPTION:
SIXMILE CREEK 74.0
END DESCRIPTION:
XS GIS Cut Line= 3
      2787405.68     10211753.12       2787593.2     10211513.59
      2787705.68     10211003.14
#Sta/Elev= 30
  4695.8 1228.22  4717.5 1226.94  4723.8  1227.4  4738.3 1224.97  4746.4 1224.54
  4759.3 1221.71  4781.7 1219.76  4831.4 1217.37  4881.2 1215.75  4924.4  1213.3
  4951.7 1210.88  4966.2 1206.72  4974.3 1203.08  4980.6 1203.24  5000.1 1202.43
  5000.6 1201.93  5020.8 1201.93  5021.3 1202.43  5030.4 1204.06  5084.4 1208.28
  5102.9 1211.33    5123 1216.12  5128.1 1215.68  5133.6 1217.11  5171.8 1216.98
  5264.4 1218.29  5379.4 1220.53  5405.8  1221.5  5481.8 1222.63  5522.7 1223.86
#Mann= 3 ,-1 , 0
  4695.8     .05       0  5000.1     .03       0  5021.3     .05       0
Bank Sta=5000.1,5021.3
XS Rating Curve= 0 ,0
Exp/Cntr=0.3,0.1

Type RM Length L Ch R = 1 ,36500   ,500,500,500
BEGIN DESCRIPTION:
SIXMILE CREEK 73.0
END DESCRIPTION:
XS GIS Cut Line= 3
      2787605.65     10211903.12      2787946.88       10211810.
       2788205.7     10211753.11
#Sta/Elev= 30
  4646.3  1222.5  4663.6 1220.48  4687.8 1220.24  4718.9 1217.05  4760.4 1215.59
  4812.1 1214.66  4874.4 1216.03  4896.8 1215.38  4905.5 1212.54  4926.1 1207.97
  4931.3 1208.08  4936.6 1206.55  4946.9 1205.87    4978 1201.37    5000 1200.47
  5000.8 1199.38  5001.3 1198.88  5021.6 1198.88  5022.1 1199.38  5029.5 1202.99
  5039.7  1205.7  5055.2 1208.06  5060.4 1206.91    5099 1209.74  5121.6 1212.66
  5142.1  1213.9    5153 1215.65  5203.6 1219.52    5224 1219.86    5265 1222.17
#Mann= 3 ,-1 , 0
  4646.3     .05       0  5000.8     .03       0  5022.1     .05       0
Bank Sta=5000.8,5022.1
XS Rating Curve= 0 ,0
Exp/Cntr=0.3,0.1

Type RM Length L Ch R = 1 ,36000   ,500,500,500
BEGIN DESCRIPTION:
SIXMILE CREEK 72.0
END DESCRIPTION:
XS GIS Cut Line= 3
      2787855.69     10212403.11      2788040.84     10212293.23
      2788305.67     10212103.12
#Sta/Elev= 30
  4784.7 1220.48  4842.8 1216.17  4924.2 1213.65  4930.9 1212.53  4951.1 1206.99
  4959.1 1204.07  4973.7 1199.79  4982.4 1199.56  4989.3 1200.07  4999.8 1199.25
  5000.3 1198.75  5020.6 1198.75  5021.1 1199.25  5025.2 1199.98  5039.9  1200.2
  5054.6 1201.15  5075.5 1206.51  5096.4 1210.09  5104.4 1210.57  5125.9 1210.11
  5161.5  1210.5  5176.2 1212.27  5190.6 1213.23  5197.1 1214.29  5232.7 1216.93
  5239.9 1218.07  5253.6 1218.68  5262.2 1218.48  5303.9 1221.13    5326 1221.85
#Mann= 4 ,-1 , 0
  4784.7     .12       0  4951.1     .05       0  4999.8     .03       0
  5021.1     .05       0
Bank Sta=4999.8,5021.1
XS Rating Curve= 0 ,0
Exp/Cntr=0.3,0.1

Type RM Length L Ch R = 1 ,35500   ,500,500,500
BEGIN DESCRIPTION:
SIXMILE CREEK 71.0
END DESCRIPTION:
XS GIS Cut Line= 3
      2788255.66     10212953.16      2788434.58     10212573.28
      2788555.69     10212203.09
#Sta/Elev= 30
  4580.1 1219.77  4639.9 1217.38  4668.6 1214.98    4746    1214  4753.8 1212.49
  4759.4 1213.02  4776.6 1211.01  4804.9 1207.07  4822.2  1209.4  4834.4  1207.6
  4856.5 1207.48  4873.3 1206.02  4889.7 1206.34  4896.1 1204.51  4901.6 1207.16
  4918.9  1204.9  4924.4 1205.71  4941.7 1201.69  4947.2 1202.22  4976.5 1197.17
    4977 1196.67  4997.9 1197.17  5031.7 1198.05  5105.4 1207.35    5158 1211.42
  5246.1 1215.31  5272.7 1217.43    5278 1216.93  5315.8 1218.71  5389.5 1223.49
#Mann= 3 ,-1 , 0
  4580.1     .05       0  4976.5     .05       0  4997.9     .05       0
Bank Sta=4976.5,4997.9
XS Rating Curve= 0 ,0
Exp/Cntr=0.3,0.1

Type RM Length L Ch R = 1 ,35000   ,500,500,500
BEGIN DESCRIPTION:
SIXMILE CREEK 70.0
END DESCRIPTION:
XS GIS Cut Line= 3
      2788655.66     10213103.15      2788839.48     10212846.74
      2789255.65     10212653.13
#Sta/Elev= 30
  4684.5 1222.59  4748.4 1220.61    4784 1217.51  4798.8 1214.15  4807.4 1213.04
    4906 1208.54  4920.4 1201.93  4935.1 1198.82  5006.8 1197.12  5018.1 1196.23
  5018.6 1195.73  5039.6 1196.23  5044.8 1197.36    5062 1197.62  5067.7 1199.74
  5096.1 1202.68  5141.8 1203.35  5159.2 1204.05  5164.7 1205.01  5187.6 1204.73
    5205 1206.12  5216.4  1208.3  5227.4 1208.36  5238.9 1209.88  5330.4 1213.92
  5359.8 1216.04  5399.1 1217.69  5404.6 1218.56  5414.9 1218.51    5459 1220.94
#Mann= 3 ,-1 , 0
  4684.5     .05       0  5018.1     .03       0  5039.6     .05       0
Bank Sta=5018.1,5039.6
XS Rating Curve= 0 ,0
Exp/Cntr=0.3,0.1

Type RM Length L Ch R = 1 ,34500   ,500,500,500
BEGIN DESCRIPTION:
SIXMILE CREEK 69.0
END DESCRIPTION:
XS GIS Cut Line= 3
      2788805.65     10213203.11      2789140.59     10213242.11
      2789255.69     10212753.08
#Sta/Elev= 30
  4662.8 1216.23  4790.6 1209.21  4879.1 1207.34  4904.5 1205.93  4922.2 1202.19
  4934.7 1197.84  4956.9 1193.46  4957.4 1192.96  4978.4 1193.46    4985 1194.94
    5000 1194.65  5009.2 1195.56  5019.5 1194.33  5038.7 1194.04  5044.6 1193.75
  5050.3 1195.95  5092.1 1201.12    5112 1201.01  5153.1 1203.89  5176.9 1203.76
  5255.8 1206.54  5261.6 1207.56  5266.8 1209.92  5286.6 1214.21    5304 1214.79
  5309.1 1216.23  5317.4 1212.37  5327.7 1210.15    5338 1210.05  5502.4 1217.42
#Mann= 5 ,-1 , 0
  4662.8     .05       0  4922.2     .12       0  4956.9     .07       0
  4978.4     .12       0  5038.7     .05       0
Bank Sta=4956.9,4978.4
XS Rating Curve= 0 ,0
Exp/Cntr=0.3,0.1

Type RM Length L Ch R = 1 ,34000   ,500,500,500
BEGIN DESCRIPTION:
SIXMILE CREEK 68.0
END DESCRIPTION:
XS GIS Cut Line= 3
      2788955.65     10214003.14      2789459.77     10213626.47
      2789855.66     10213103.14
#Sta/Elev= 30
  4370.7 1242.19  4413.5 1238.37  4428.1  1234.7  4434.3 1236.27  4442.7 1234.47
  4448.9 1235.92  4463.5 1233.29  4478.1 1228.51  4484.3 1229.89  4492.7 1228.18
  4498.9 1228.87  4534.4  1223.4  4634.4 1216.92  4657.4 1213.92  4734.5  1212.3
  4770.2 1208.86  4836.4 1206.05  4913.7 1203.27  4963.8 1193.25    4993 1194.12
  5017.9 1192.67  5018.4 1192.17  5039.8 1192.67  5070.5 1198.62    5092 1198.74
  5128.7 1202.39  5378.4 1206.19  5584.5 1212.07    5599 1213.71  5656.2 1214.22
#Mann= 5 ,-1 , 0
  4370.7     .05       0  4836.4     .12       0  4963.8     .05       0
  5017.9     .03       0  5039.8     .05       0
Bank Sta=5017.9,5039.8
XS Rating Curve= 0 ,0
Exp/Cntr=0.3,0.1

Type RM Length L Ch R = 1 ,33500   ,500,500,500
BEGIN DESCRIPTION:
SIXMILE CREEK 67.0
END DESCRIPTION:
XS GIS Cut Line= 3
      2789405.69     10214453.11      2789733.73     10214042.96
      2790005.69     10213553.09
#Sta/Elev= 30
  4474.8 1228.32    4546 1221.86  4581.3  1217.6  4638.9 1215.39  4659.7 1213.23
  4674.1 1215.16  4694.9 1211.99  4717.3 1213.13  4758.9  1212.3  4781.4 1207.88
  4787.8    1208  4794.9 1206.15    4823 1202.81  4909.4 1201.91  4915.8 1199.57
  4930.2 1197.85  4936.6 1194.32  4944.6 1193.48  4954.4 1189.18  4954.9 1188.68
  4976.4 1189.18  5053.4 1192.17  5059.1 1194.86  5075.2 1198.03  5080.9 1200.76
  5102.8 1204.81  5205.7 1203.05  5274.3 1203.71  5384.1 1207.16  5560.3 1214.66
#Mann= 3 ,-1 , 0
  4474.8     .05       0  4954.4     .05       0  4976.4     .05       0
Bank Sta=4954.4,4976.4
XS Rating Curve= 0 ,0
Exp/Cntr=0.3,0.1

Type RM Length L Ch R = 1 ,33000   ,500,500,500
BEGIN DESCRIPTION:
SIXMILE CREEK 66.0
END DESCRIPTION:
XS GIS Cut Line= 3
      2789555.72      10214503.1      2790063.25       10214397.
      2790305.69      10213903.1
#Sta/Elev= 30
  4481.5 1216.86  4532.5 1211.17  4624.5 1209.88  4656.4  1207.6  4675.6  1207.7
  4736.9  1202.4  4777.7 1201.77  4801.2 1199.36  4828.8 1199.57  4846.1 1196.67
  4851.2  1198.9  4879.9 1194.12    4896 1195.53  4901.1 1194.05    4946 1189.57
  4960.8 1189.25  4961.3 1188.75  4982.8 1189.25    4996 1190.87  5041.4 1191.17
  5063.9 1196.01  5071.2 1199.97  5086.4 1201.75  5148.3 1199.75  5182.6 1199.91
  5198.9 1196.06  5215.8 1199.16  5238.3  1200.5  5371.9 1203.76  5550.2 1211.59
#Mann= 3 ,-1 , 0
  4481.5     .05       0  4960.8     .05       0  4982.8     .05       0
Bank Sta=4960.8,4982.8
XS Rating Curve= 0 ,0
Exp/Cntr=0.3,0.1

Type RM Length L Ch R = 1 ,32500   ,500,500,500
BEGIN DESCRIPTION:
SIXMILE CREEK 65.0
END DESCRIPTION:
XS GIS Cut Line= 3
      2790205.65     10214903.15      2790550.02      10214486.3
      2790955.69     10214003.11
#Sta/Elev= 30
  4459.3 1209.16  4672.3 1200.54  4715.3 1199.99  4721.8 1199.14  4729.7 1199.89
  4828.7 1198.19  4849.5 1196.93  4863.8 1194.93  4871.7 1190.33  4878.2 1189.07
  4906.8 1190.18  4927.7 1188.69    4942 1189.11  4967.1 1188.11  4967.6 1187.61
  4989.3 1188.11  4991.5 1188.79  5020.2 1188.55  5034.5 1191.11  5048.8 1196.73
  5063.1 1193.98  5069.6 1195.16  5077.4 1195.18  5083.9 1197.13  5098.2 1197.85
    5184 1200.05    5361 1206.82  5410.4 1210.06  5496.2 1213.51  5630.9  1221.3
#Mann= 3 ,-1 , 0
  4459.3     .05       0  4967.1     .03       0  4989.3     .05       0
Bank Sta=4967.1,4989.3
XS Rating Curve= 0 ,0
Exp/Cntr=0.3,0.1

Type RM Length L Ch R = 1 ,32000   ,500,500,500
BEGIN DESCRIPTION:
SIXMILE CREEK 64.0
END DESCRIPTION:
XS GIS Cut Line= 3
      2790455.71      10215153.1      2790820.87     10214899.47
      2791055.69     10214703.11
#Sta/Elev= 30
  4555.4 1210.19  4568.9  1210.6  4598.6 1207.34  4713.7 1202.26  4762.7  1198.4
  4798.9 1196.54  4899.8 1197.95  4914.6 1195.84  4929.5  1191.9  4944.3  1189.2
  4971.4 1187.78  4988.8 1185.05  4989.3 1184.55    5011 1185.05  5029.6 1185.96
  5036.1 1185.54  5064.7 1188.31  5071.5    1191    5079 1190.19  5093.3  1191.9
  5099.8  1191.5  5142.8 1194.22  5163.6 1200.05  5177.9 1201.93  5205.8  1203.6
    5256 1206.45  5265.4 1206.11  5278.1 1206.62  5284.6 1207.83  5306.1  1208.1
#Mann= 5 ,-1 , 0
  4555.4     .05       0  4988.8     .03       0    5011     .05       0
  5205.8     .12       0  5265.4     .05       0
Bank Sta=4988.8,5011
XS Rating Curve= 0 ,0
Exp/Cntr=0.3,0.1

Type RM Length L Ch R = 1 ,31500   ,500,500,500
BEGIN DESCRIPTION:
SIXMILE CREEK 63.0
END DESCRIPTION:
XS GIS Cut Line= 3
      2790505.71     10215453.11      2791007.07     10215360.73
      2791405.67     10215003.13
#Sta/Elev= 30
  4490.2    1210  4516.7 1207.86    4541 1207.55  4569.7 1206.15    4602 1205.86
  4627.8 1203.79  4733.8 1199.65  4791.9 1196.11    4850 1194.67  4876.6 1190.82
  4917.2 1186.46  5035.8 1184.37  5036.3 1183.87  5057.7 1183.87  5058.2 1184.37
  5061.2  1190.5  5067.9 1189.52  5075.4 1195.29  5140.1 1195.45  5157.1 1195.55
  5195.8  1196.5  5202.5 1195.95  5216.7 1196.31  5266.8 1198.29  5280.3 1199.75
  5315.5  1200.5  5408.1 1203.59  5453.5 1205.91  5528.4 1206.43  5535.5 1207.09
#Mann= 7 ,-1 , 0
  4490.2     .05       0  5035.8     .03       0  5058.2     .05       0
  5140.1     .12       0  5157.1     .05       0  5315.5     .12       0
  5453.5     .05       0
Bank Sta=5035.8,5058.2
XS Rating Curve= 0 ,0
Exp/Cntr=0.3,0.1

Type RM Length L Ch R = 1 ,31000   ,500,500,500
BEGIN DESCRIPTION:
SIXMILE CREEK 62.0
END DESCRIPTION:
XS GIS Cut Line= 3
      2791055.69      10216053.1      2791266.27     10215781.47
       2791655.7      10215453.1
#Sta/Elev= 30
  4656.3 1209.21  4692.5 1206.09  4713.3 1203.35  4770.2 1199.58  4812.9 1198.28
  4820.8  1197.6  4827.4  1196.1  4833.7    1196  4848.2 1193.49  4877.2 1191.54
    4884 1192.11  4891.7 1191.51  4941.5 1182.89  4955.9 1184.22  4991.2 1183.05
  4994.2 1182.37  4994.7 1181.87  5016.8 1182.37  5048.4 1186.16    5077 1188.19
  5090.8  1187.9  5126.4 1189.54  5147.2  1192.3    5155 1192.03  5175.8 1194.67
    5211 1197.66  5389.1  1205.2  5438.5 1205.76  5481.4 1208.76  5509.4 1209.87
#Mann= 3 ,-1 , 0
  4656.3     .05       0  4994.2     .05       0  5016.8     .05       0
Bank Sta=4994.2,5016.8
XS Rating Curve= 0 ,0
Exp/Cntr=0.3,0.1

Type RM Length L Ch R = 1 ,30500   ,500,500,500
BEGIN DESCRIPTION:
SIXMILE CREEK 61.0
END DESCRIPTION:
XS GIS Cut Line= 3
      2791405.67     10216353.12      2791627.17      10216125.1
       2792005.7     10215603.09
#Sta/Elev= 30
  4682.1 1206.88  4696.2 1205.05  4703.3 1202.77  4724.5 1199.44  4745.8 1198.13
  4752.7 1196.57  4766.9  1195.3  4802.7 1194.19  4883.9  1190.6  4908.4 1189.74
  4915.5 1187.98  4929.7  1180.7  4939.5 1180.59    4940 1180.09  4962.1 1180.59
  4964.9 1181.82  4986.3 1181.46  5028.2 1184.21  5051.4 1183.53  5122.5 1188.59
  5137.2    1191  5143.4 1193.02  5150.7 1193.52  5308.8 1198.08    5315 1199.12
  5365.3 1198.74  5400.8 1200.58  5495.2 1201.69  5572.5 1205.91  5644.8 1208.62
#Mann= 5 ,-1 , 0
  4682.1     .12       0  4802.7     .05       0  4883.9     .12       0
  4939.5     .03       0  4962.1     .05       0
Bank Sta=4939.5,4962.1
XS Rating Curve= 0 ,0
Exp/Cntr=0.3,0.1

Type RM Length L Ch R = 1 ,30000   ,500,500,500
BEGIN DESCRIPTION:
SIXMILE CREEK 60.0
END DESCRIPTION:
XS GIS Cut Line= 3
      2791755.68     10216903.11       2791948.8     10216506.31
      2792205.66     10216303.13
#Sta/Elev= 30
  4558.7 1213.23  4662.9 1203.92  4679.9 1203.36  4714.4 1199.82    4770 1196.15
  4781.2 1194.25  4814.5 1193.75  4820.8 1191.96  4826.3 1192.03  4848.9 1188.61
    4859 1188.87  4888.4 1185.89  4925.7  1184.5  4947.9 1179.65  4961.6 1178.05
  4981.1 1177.84  4981.6 1177.34  5003.8 1177.84  5028.6 1180.63  5043.1 1184.12
  5078.3  1187.4  5092.7 1190.48  5107.2 1191.83  5113.5 1193.68    5136 1189.22
  5162.4 1189.53  5235.4  1193.3  5270.6 1196.79  5292.8 1197.79  5327.5 1198.73
#Mann= 5 ,-1 , 0
  4558.7     .05       0  4981.1     .05       0  5003.8     .05       0
  5162.4     .12       0  5292.8     .05       0
Bank Sta=4981.1,5003.8
XS Rating Curve= 0 ,0
Exp/Cntr=0.3,0.1

Type RM Length L Ch R = 1 ,29500   ,500,500,500
BEGIN DESCRIPTION:
SIXMILE CREEK 59.0
END DESCRIPTION:
XS GIS Cut Line= 3
      2792005.69     10216903.11      2792333.85     10216822.56
      2792755.67     10216753.11
#Sta/Elev= 30
  4662.1 1198.84  4768.6 1193.07  4785.7 1190.61    4805 1189.95  4810.2 1187.49
  4826.8 1185.25  4898.9 1182.69  4934.9 1180.15  4960.7 1177.37  5003.5 1177.34
  5015.9 1176.52  5016.4 1176.02  5038.7 1176.52  5042.4 1179.33  5052.5  1181.6
  5062.7 1183.35  5082.9 1184.12  5093.5 1186.14  5113.3 1186.51  5123.5 1185.52
  5141.3 1181.37  5149.7 1178.59  5154.7 1180.06    5164 1179.73  5174.1 1183.09
  5184.3 1184.72  5210.8 1187.04  5326.2 1192.16  5385.9 1196.15  5427.5 1198.79
#Mann= 5 ,-1 , 0
  4662.1     .05       0  5015.9     .05       0  5038.7     .05       0
  5141.3     .12       0  5385.9     .05       0
Bank Sta=5015.9,5038.7
XS Rating Curve= 0 ,0
Exp/Cntr=0.3,0.1

Type RM Length L Ch R = 1 ,29000   ,500,500,500
BEGIN DESCRIPTION:
SIXMILE CREEK 58.0
END DESCRIPTION:
XS GIS Cut Line= 3
      2792305.69     10217303.11      2792660.12     10217185.93
      2793055.72     10216853.08
#Sta/Elev= 30
  4626.7 1198.08  4737.7  1193.9  4795.2 1191.38  4838.2 1188.46  4858.4 1188.09
  4869.9 1186.56    4890 1185.16  4901.6 1183.17  4953.2 1180.08  4974.3 1177.02
  4984.8 1176.98  4991.6 1176.24    5000 1176.48  5008.9 1175.44  5009.4 1174.94
  5031.3 1174.94  5031.8 1175.44  5062.4 1177.08  5076.7 1179.76  5111.8 1184.08
  5169.1 1186.87  5190.2 1186.88  5247.1 1189.36  5353.7 1197.25  5382.3 1198.87
  5403.2 1198.95  5446.1 1202.31  5452.6  1202.3  5460.4 1203.37    5517 1206.83
#Mann= 3 ,-1 , 0
  4626.7     .05       0  5008.9     .03       0  5031.8     .05       0
Bank Sta=5008.9,5031.8
XS Rating Curve= 0 ,0
Exp/Cntr=0.3,0.1

Type RM Length L Ch R = 1 ,28500   ,500,500,500
BEGIN DESCRIPTION:
SIXMILE CREEK 57.0
END DESCRIPTION:
XS GIS Cut Line= 3
      2792755.72     10217703.09        2792936.      10217595.4
      2793355.68     10217103.11
#Sta/Elev= 30
    4790 1195.15    4825 1191.57  4840.5 1191.21  4856.1 1188.61  4861.9 1188.64
  4906.4 1183.46  4951.5 1180.89  4972.9 1175.24  4982.8 1173.76  4983.3 1173.26
  5005.7 1173.76  5008.4 1175.13  5016.1 1175.39  5051.2 1174.39  5065.5 1175.13
  5094.1 1177.21  5135.8 1182.12  5213.7 1187.03  5235.7 1187.32  5278.5 1189.94
  5292.1 1189.97  5299.4 1191.04  5426.7 1196.29  5469.6  1200.1  5490.4 1200.99
  5498.1 1202.22  5504.7 1201.88  5533.2 1203.73  5561.8 1206.86  5646.9 1211.67
#Mann= 3 ,-1 , 0
    4790     .05       0  4982.8     .03       0  5005.7     .05       0
Bank Sta=4982.8,5005.7
XS Rating Curve= 0 ,0
Exp/Cntr=0.3,0.1

Type RM Length L Ch R = 1 ,28000   ,500,500,500
BEGIN DESCRIPTION:
SIXMILE CREEK 56.0
END DESCRIPTION:
XS GIS Cut Line= 3
      2792755.67     10217953.11      2793230.91     10217997.45
      2793355.67     10217653.16
#Sta/Elev= 30
  4522.7 1206.79  4577.2 1204.57  4613.1 1201.75  4623.1 1202.02  4681.3 1194.77
  4753.7 1190.36  4790.3 1186.59  4795.4 1186.91    4814 1185.75  4844.1 1181.75
  4884.3 1178.84  4899.4 1176.95  4904.4 1177.72  4934.5 1173.96  4964.6 1173.01
  4973.3 1171.13  4973.8 1170.63  4996.2 1171.13  4999.9 1172.26  5055.3  1173.6
  5060.6 1174.84  5085.9 1177.12  5091.2 1178.58  5141.8 1181.44  5147.2 1182.52
  5177.8 1184.69  5217.3 1185.38  5233.7 1184.97  5264.4 1187.71  5366.2 1192.83
#Mann= 3 ,-1 , 0
  4522.7     .05       0  4973.3     .05       0  4996.2     .05       0
Bank Sta=4973.3,4996.2
XS Rating Curve= 0 ,0
Exp/Cntr=0.3,0.1

Type RM Length L Ch R = 1 ,27500   ,500,500,500
BEGIN DESCRIPTION:
SIXMILE CREEK 55.0
END DESCRIPTION:
XS GIS Cut Line= 3
       2793205.7     10218553.11      2793414.23     10218457.74
      2793805.67     10218253.12
#Sta/Elev= 30
  4770.7 1192.42  4859.5 1182.03  4905.5 1179.73  4928.6  1177.5  4951.6 1174.42
  4967.6 1170.11  4968.1 1169.61  4992.1 1169.61  4992.6 1170.11  5035.5  1170.8
  5063.8 1173.87  5085.9    1175  5114.5 1178.95  5159.6 1182.76  5196.3 1184.54
  5212.7 1186.36  5218.4 1185.63  5256.9 1185.91  5262.5 1186.72  5272.5 1186.14
    5301 1186.52  5306.7 1187.65  5328.9 1187.37  5339.6 1187.69  5345.2 1188.57
  5361.6  1188.8  5367.3 1189.64  5383.7 1189.52  5405.8 1191.01  5441.7  1191.4
#Mann= 3 ,-1 , 0
  4770.7     .05       0  4967.6     .05       0  4992.6     .05       0
Bank Sta=4967.6,4992.6
XS Rating Curve= 0 ,0
Exp/Cntr=0.3,0.1

Type RM Length L Ch R = 1 ,27000   ,500,500,500
BEGIN DESCRIPTION:
SIXMILE CREEK 54.0
END DESCRIPTION:
XS GIS Cut Line= 3
      2793305.67     10218903.11      2793530.24     10218941.91
      2793905.72     10219053.12
#Sta/Elev= 30
  4772.1  1191.7  4799.5 1189.56  4804.6 1189.97  4812.7 1189.42  4843.2 1186.27
  4883.7 1183.09    4914 1175.37  4919.1 1176.32  4924.3 1173.91  4934.5 1170.88
  4954.8 1169.09  4982.6 1168.31  4983.1 1167.81  5007.2 1167.81  5007.7 1168.31
  5026.8 1169.48  5054.8 1173.69    5060 1173.41  5068.3 1174.57  5093.3 1174.44
  5099.5 1173.87    5193 1177.76  5236.7 1178.71  5245.6 1180.19    5270 1181.22
  5276.8 1182.45  5303.2 1184.79  5308.4 1184.33  5360.3 1187.93  5391.6 1190.86
#Mann= 3 ,-1 , 0
  4772.1     .05       0  4982.6     .03       0  5007.7     .05       0
Bank Sta=4982.6,5007.7
XS Rating Curve= 0 ,0
Exp/Cntr=0.3,0.1

Type RM Length L Ch R = 1 ,26500   ,500,500,500
BEGIN DESCRIPTION:
SIXMILE CREEK 53.0
END DESCRIPTION:
XS GIS Cut Line= 3
      2793355.65     10219503.12      2793711.75      10219406.8
      2793955.71     10219353.11
#Sta/Elev= 30
  4631.1 1192.15  4728.2 1187.61  4768.1 1184.79  4796.9 1181.82  4802.8 1180.19
    4808 1180.35  4837.5 1177.75  4848.7 1177.32  4869.4 1178.23  4890.1 1173.77
  4931.6 1170.09  4951.9 1166.38  4979.2 1165.98  4979.7 1165.48  5004.3 1165.98
  5004.6 1167.49  5014.3 1166.98  5024.5 1168.05  5034.7 1169.76  5045.3 1172.83
  5083.9 1178.88    5089 1178.23  5106.4 1181.08  5126.9 1182.46  5132.7 1184.23
  5149.5 1185.31  5182.6 1187.39  5198.6 1189.19  5225.3 1189.71  5249.8 1191.72
#Mann= 5 ,-1 , 0
  4631.1     .05       0  4979.2     .03       0  5004.3     .05       0
  5149.5     .12       0  5182.6     .05       0
Bank Sta=4979.2,5004.3
XS Rating Curve= 0 ,0
Exp/Cntr=0.3,0.1

Type RM Length L Ch R = 1 ,26000   ,500,500,500
BEGIN DESCRIPTION:
SIXMILE CREEK 52.0
END DESCRIPTION:
XS GIS Cut Line= 3
      2793355.67      10219653.1       2793687.1     10219871.64
      2793805.71     10219953.13
#Sta/Elev= 30
    4603 1189.73  4703.9 1181.23  4724.9 1177.83  4761.1 1174.87  4818.6 1173.24
  4833.3 1174.97  4863.5 1174.78  4878.5 1173.41  4905.6 1167.92  4937.7 1163.52
  4938.2 1163.02  4962.6 1163.02  4963.1 1163.52  4971.9  1164.5    4993 1164.07
  5007.9 1165.02    5014 1166.59  5022.5 1167.65  5025.4  1169.1  5034.9 1173.37
  5043.7 1178.27  5049.8 1179.91  5060.2 1181.45  5071.1 1184.01  5085.7 1185.41
  5107.5 1189.04  5115.5 1188.93  5136.4 1190.39  5140.8 1191.91  5143.9 1191.91
#Mann= 5 ,-1 , 0
    4603     .05       0  4937.7     .05       0  4963.1     .05       0
  5025.4     .12       0  5060.2     .05       0
Bank Sta=4937.7,4963.1
XS Rating Curve= 0 ,0
Exp/Cntr=0.3,0.1

Type RM Length L Ch R = 1 ,25500   ,668,668,668
BEGIN DESCRIPTION:
SIXMILE CREEK 51.0
END DESCRIPTION:
XS GIS Cut Line= 3
      2793155.69     10219653.14      2793215.62     10219990.05
       2793305.7     10220253.16
#Sta/Elev= 30
  4657.8 1193.08  4728.9 1189.32  4743.8 1188.19  4779.7 1183.58  4797.7 1181.98
  4802.8 1182.58  4830.4 1176.43  4856.7 1174.31  4881.2 1173.46  4910.7 1168.81
  4915.8 1169.11  4921.9 1166.84  4980.3 1161.84  4980.8 1161.34  5005.7 1161.84
  5024.4 1162.44  5034.9 1163.68  5043.4 1165.94  5048.7 1165.87  5056.1 1167.09
  5111.2 1169.77  5137.2 1175.11  5161.8 1177.07  5168.5 1178.61  5214.6 1183.77
  5231.1 1190.18  5240.3  1190.6  5246.3 1191.41  5262.4 1190.97  5278.1 1192.87
#Mann= 4 ,-1 , 0
  4657.8     .05       0  4980.3     .05       0  5005.7     .05       0
  5240.3     .12       0
Bank Sta=4980.3,5005.7
XS Rating Curve= 0 ,0
Exp/Cntr=0.3,0.1

Type RM Length L Ch R = 1 ,24832   ,332,332,332
BEGIN DESCRIPTION:
Mapping XS c1aa224d
END DESCRIPTION:
XS GIS Cut Line= 4
      2792467.01      10219542.7      2792555.56     10219850.03
      2792565.98     10220230.23      2792638.89     10220443.75
#Sta/Elev= 30
  4427.4 1186.19  4615.2 1184.87    4688 1180.61  4708.8 1178.41    4740 1176.86
  4746.2  1175.5  4850.4 1170.44  4870.4  1168.1  4880.4 1168.25  4900.4 1164.44
  4910.4 1164.13  4929.8 1159.87  4934.8 1159.87  4940.4 1161.47  4997.7 1157.62
  4998.2 1157.12  5023.2 1157.62  5030.4 1161.01  5050.4 1166.73  5100.4 1179.14
  5120.5  1182.5  5126.5 1184.84  5131.7 1184.84  5151.8 1188.62  5183.5 1192.56
  5246.9    1196  5264.3 1197.96  5289.1 1197.56    5342 1198.86  5353.2 1198.15
#Mann= 3 ,-1 , 0
  4427.4     .05       0  4997.7     .05       0  5023.2     .05       0
Bank Sta=4997.7,5023.2
XS Rating Curve= 0 ,0
Exp/Cntr=0.3,0.1

Type RM Length L Ch R = 1 ,24500   ,500,500,500
BEGIN DESCRIPTION:
SIXMILE CREEK 49.0
END DESCRIPTION:
XS GIS Cut Line= 3
      2792355.67     10219853.15      2792248.11     10220187.16
      2792355.69     10220453.12
#Sta/Elev= 30
  4649.1 1179.29  4675.9 1178.24  4754.1 1174.76  4775.1 1173.53  4793.4 1171.52
  4830.7 1170.48  4857.5 1168.09  4862.8 1168.49  4889.6 1166.19  4926.9  1164.3
  4932.7 1162.16  4953.7 1162.14  4964.2 1159.27  5020.7  1157.7  5021.2  1157.2
  5046.2  1157.7  5057.6 1161.36  5071.1 1163.86  5111.2 1165.47  5157.4 1169.56
    5189  1173.3  5211.4 1177.75  5218.5 1178.11    5233 1180.59  5242.6 1183.77
    5248 1186.91  5254.5 1187.54  5272.1 1186.51  5277.5 1189.48  5286.9 1190.17
#Mann= 4 ,-1 , 0
  4649.1     .12       0  4675.9     .05       0  5020.7     .05       0
  5046.2     .05       0
Bank Sta=5020.7,5046.2
XS Rating Curve= 0 ,0
Exp/Cntr=0.3,0.1

Type RM Length L Ch R = 1 ,24000   ,500,500,500
BEGIN DESCRIPTION:
SIXMILE CREEK 48.0
END DESCRIPTION:
XS GIS Cut Line= 3
       2791605.7     10220153.13      2791786.77     10220347.31
      2791755.68     10220603.12
#Sta/Elev= 30
  4734.5 1180.85  4737.9 1180.85  4755.7 1184.27  4776.7 1174.04  4798.2 1169.75
  4805.1 1169.89  4869.1 1165.57  4875.9 1165.89  4925.7 1162.93  4932.6 1163.12
  4946.7  1161.6  4953.6 1161.73  4960.9 1160.24  4967.8 1161.14  4975.1 1158.21
  4981.9 1159.44  4989.3 1156.99  5015.9 1156.41  5036.1 1157.92  5045.8 1157.76
  5056.2 1156.92  5063.5 1155.09    5064 1154.59  5089.2 1155.09  5106.6 1161.63
  5126.7 1165.71  5137.6 1171.36    5157 1169.64    5167 1170.06  5257.7 1178.99
#Mann= 3 ,-1 , 0
  4734.5     .05       0  5063.5     .03       0  5089.2     .05       0
Bank Sta=5063.5,5089.2
XS Rating Curve= 0 ,0
Exp/Cntr=0.3,0.1

Type RM Length L Ch R = 1 ,23500   ,500,500,500
BEGIN DESCRIPTION:
SIXMILE CREEK 47.0
END DESCRIPTION:
XS GIS Cut Line= 3
      2791255.69     10220153.13      2791315.33     10220486.23
      2791255.68     10220753.15
#Sta/Elev= 30
  4661.6 1178.76  4747.3 1174.37  4763.2 1175.29  4773.3 1177.74  4783.5 1176.77
  4793.7  1174.8  4801.1 1171.88  4806.2 1171.51    4814 1166.74  4824.1 1162.15
  4844.4 1159.35  4859.9  1155.4  4874.9 1154.29    4946  1156.8  4966.4 1156.37
  4977.6 1155.31    4983  1152.4  4983.5  1151.9  5008.7  1152.4  5021.9 1153.93
  5036.4 1157.94  5058.3 1161.23  5099.3 1164.86  5113.8 1167.51  5119.8 1169.65
  5150.5 1169.53    5171 1172.51    5212 1176.58  5232.5 1177.62  5273.5 1182.44
#Mann= 4 ,-1 , 0
  4661.6     .05       0    4983     .05       0  5008.7     .05       0
  5036.4     .12       0
Bank Sta=4983,5008.7
XS Rating Curve= 0 ,0
Exp/Cntr=0.3,0.1

Type RM Length L Ch R = 1 ,23000   ,500,500,500
BEGIN DESCRIPTION:
SIXMILE CREEK 46.0
END DESCRIPTION:
XS GIS Cut Line= 3
      2790755.69     10220203.16      2790824.01     10220529.38
      2791055.68     10220803.11
#Sta/Elev= 30
  4666.7 1176.03    4728 1174.19  4736.4 1172.53  4741.6 1172.62  4748.4 1170.49
    4779 1168.44  4809.7 1163.81  4922.1  1157.6  4942.5 1153.71  4962.9 1152.16
  4973.2 1149.28  4973.7 1148.78    4999 1149.28  4999.4 1150.02  5010.9 1149.76
    5018 1150.41  5025.2 1153.11  5031.7 1154.41  5039.5 1158.83    5046  1158.5
  5060.3 1161.77  5144.5  1165.9  5166.9 1167.09  5195.5 1171.34  5209.8 1171.52
    5224 1173.26  5230.6 1172.93  5259.2 1174.45    5280 1176.45  5358.6 1180.63
#Mann= 4 ,-1 , 0
  4666.7     .05       0  4973.2     .05       0    4999     .05       0
  5144.5     .12       0
Bank Sta=4973.2,4999
XS Rating Curve= 0 ,0
Exp/Cntr=0.3,0.1

Type RM Length L Ch R = 1 ,22500   ,500,500,500
BEGIN DESCRIPTION:
SIXMILE CREEK 45.0
END DESCRIPTION:
XS GIS Cut Line= 3
      2790205.67     10220403.09      2790391.74     10220766.31
      2790655.73     10220853.13
#Sta/Elev= 30
  4591.9 1176.01  4605.8  1174.6  4622.4 1169.62  4644.6 1168.46  4672.4 1168.59
  4711.2  1165.2  4716.8 1165.82  4733.4  1164.7  4749.2    1165  4777.8 1162.01
  4786.6 1161.91  4805.7 1160.91  4816.6 1162.75  4828.9 1159.44  4883.2  1157.7
  4899.5 1158.42    4911 1158.73  4927.6 1157.65  4955.5 1153.83  4962.7 1151.53
  4977.7 1148.65  5001.7 1147.99  5002.2 1147.49  5027.6 1147.99  5034.1 1148.34
  5060.2 1153.13  5077.8 1156.31  5134.8 1159.84  5235.7 1169.31  5277.9 1171.71
#Mann= 7 ,-1 , 0
  4591.9     .05       0  4786.6     .12       0  4828.9     .05       0
  4899.5     .12       0  5001.7     .07       0  5027.6     .12       0
  5060.2     .05       0
Bank Sta=5001.7,5027.6
XS Rating Curve= 0 ,0
Exp/Cntr=0.3,0.1

Type RM Length L Ch R = 1 ,22000   ,500,500,500
BEGIN DESCRIPTION:
SIXMILE CREEK 44.0
END DESCRIPTION:
XS GIS Cut Line= 3
      2789655.69     10220703.11      2789981.58     10221049.92
      2790255.66     10221453.08
#Sta/Elev= 30
  4524.1 1175.73    4538 1176.06  4665.5  1171.2  4679.7 1171.97  4701.1  1169.9
  4715.3  1169.9    4814 1164.85  4835.5 1162.54  4885.9 1160.01  4969.8 1152.89
  4976.9 1150.27    4992 1148.49  4992.5 1147.99  5017.9 1148.49  5019.1 1150.12
  5040.1 1148.69  5063.9 1150.05  5076.4 1149.43  5084.9 1150.94  5099.8 1150.75
  5112.7 1153.85  5171.7 1156.49  5185.2    1159  5192.7 1161.59  5234.6  1161.5
  5262.3  1163.1  5279.5 1164.57  5336.4 1165.92  5438.1 1174.27  5487.5 1177.12
#Mann= 5 ,-1 , 0
  4524.1     .05       0  4885.9     .12       0    4992     .07       0
  5017.9     .12       0  5262.3     .12       0
Bank Sta=4992,5017.9
XS Rating Curve= 0 ,0
Exp/Cntr=0.3,0.1

Type RM Length L Ch R = 1 ,21500   ,500,500,500
BEGIN DESCRIPTION:
SIXMILE CREEK 43.0
END DESCRIPTION:
XS GIS Cut Line= 3
      2789305.72     10221203.13      2789664.64     10221426.02
      2790055.68     10221653.11
#Sta/Elev= 30
  4577.5  1172.8  4679.6 1164.93  4700.9  1165.4  4716.2 1161.97  4722.1 1163.14
  4737.5 1159.52  4751.3 1159.11    4832    1151  4883.5 1150.74  4889.8 1148.68
  4926.4 1147.39  4947.7 1148.34    4950 1142.97  4950.5 1142.47  4976.1 1142.97
  4977.7 1146.93  4984.3 1147.52  5002.1 1145.59  5005.6 1143.53  5027.1 1148.47
  5085.9 1148.71  5138.9 1155.42  5144.7 1152.95  5166.2 1153.95  5181.9 1156.94
  5246.5 1161.66    5279 1168.16  5290.3  1170.3  5358.3 1170.54  5452.2 1172.36
#Mann= 6 ,-1 , 0
  4577.5     .12       0  4751.3     .05       0    4950     .05       0
  4976.1     .05       0    5279     .12       0  5358.3     .05       0
Bank Sta=4950,4976.1
XS Rating Curve= 0 ,0
Exp/Cntr=0.3,0.1

Type RM Length L Ch R = 1 ,21000   ,500,500,500
BEGIN DESCRIPTION:
SIXMILE CREEK 42.0
END DESCRIPTION:
XS GIS Cut Line= 3
       2789105.7     10221653.12      2789455.54     10221829.97
       2789705.7     10221803.11
#Sta/Elev= 30
    4608 1169.59  4621.9 1166.88  4638.6 1166.32  4644.2 1164.88  4683.2 1162.02
  4688.8 1160.57    4720 1158.46  4727.8 1158.89  4733.4  1157.4  4742.4 1158.28
  4800.4  1150.4  4839.2 1146.42  4861.5 1146.35  4867.1 1145.19  4883.8 1147.47
  4889.4 1145.94  4911.7 1144.37  4928.4 1138.53    4934 1139.42  4950.7 1135.71
  4995.2 1135.69  5003.2  1134.8  5003.7  1134.3  5029.3  1134.8  5040.4  1135.4
  5060.5 1140.09  5100.7 1143.68  5113.4 1143.75  5191.2 1152.54  5251.6 1156.06
#Mann= 4 ,-1 , 0
    4608     .12       0  4800.4     .05       0  5003.2     .05       0
  5029.3     .05       0
Bank Sta=5003.2,5029.3
XS Rating Curve= 0 ,0
Exp/Cntr=0.3,0.1

Type RM Length L Ch R = 1 ,20500   ,500,500,500
BEGIN DESCRIPTION:
SIXMILE CREEK 41.0
END DESCRIPTION:
XS GIS Cut Line= 3
      2788955.71     10222403.11      2789447.67     10222327.71
       2789855.7     10222253.11
#Sta/Elev= 30
  4502.3 1162.65  4545.1 1159.85  4595.6  1156.4  4674.3 1153.18  4714.7  1153.3
  4745.1 1151.28  4777.9 1151.46    4795 1152.23    4800 1151.16  4815.9 1151.35
  4886.7 1147.55  4896.8 1145.34  4906.9 1144.51  4917.1 1141.24  4926.7 1139.63
  4947.4 1137.99  4967.6 1137.93    4995 1133.69  4995.5 1133.19  5021.2 1133.69
  5028.5 1134.54    5059 1134.06  5099.6 1135.11  5111.9 1136.22  5130.1 1139.49
  5150.5 1141.88  5223.4 1148.35  5276.7 1151.27  5329.9 1156.45  5414.8  1160.4
#Mann= 6 ,-1 , 0
  4502.3     .12       0  4545.1     .05       0  4595.6     .12       0
  4777.9     .05       0    4995     .05       0  5021.2     .05       0
Bank Sta=4995,5021.2
XS Rating Curve= 0 ,0
Exp/Cntr=0.3,0.1

Type RM Length L Ch R = 1 ,20000   ,500,500,500
BEGIN DESCRIPTION:
SIXMILE CREEK 40.0
END DESCRIPTION:
XS GIS Cut Line= 3
      2789255.68      10222453.1      2789463.43     10222789.64
      2789705.69     10222753.11
#Sta/Elev= 30
  4604.5 1152.37  4612.8 1150.97  4728.1 1142.16  4749.4 1139.05  4764.7 1138.79
    4786 1134.14  4801.4 1133.01  4822.7 1132.62    4844 1135.96  4865.2 1136.62
  4901.9 1133.41  4917.3 1133.82  4923.2  1135.2  4932.7 1133.73  4953.9 1133.83
  4968.8 1132.23  4981.1 1127.88  4996.5 1127.73  5000.7 1125.88  5001.2 1125.38
  5026.9 1125.88  5032.6 1130.34  5042.7 1135.14  5077.7 1138.06  5093.3 1144.22
  5141.6 1152.58    5154 1156.69  5194.4 1156.04  5234.9 1160.89    5245 1160.74
#Mann= 4 ,-1 , 0
  4604.5     .12       0  4612.8     .05       0  5000.7     .05       0
  5026.9     .05       0
Bank Sta=5000.7,5026.9
XS Rating Curve= 0 ,0
Exp/Cntr=0.3,0.1

Type RM Length L Ch R = 1 ,19500   ,618,618,618
BEGIN DESCRIPTION:
SIXMILE CREEK 39.0
END DESCRIPTION:
XS GIS Cut Line= 3
      2788955.69     10222653.14      2789017.37     10222838.66
      2789105.68      10223103.1
#Sta/Elev= 30
  4804.5 1151.78  4846.6 1146.51    4852 1144.48  4857.2 1144.59  4867.7 1142.87
  4883.6 1138.33  4915.3 1134.33  4930.9 1133.78  4941.5 1131.93  4946.9 1128.87
  4962.5  1128.4  4973.1 1125.93  4978.6 1122.65  4983.8 1122.36  4986.6 1118.91
  4987.1 1118.41  5012.8 1118.91  5047.1  1125.3    5068 1126.17    5089 1129.52
  5110.3  1131.6  5120.7 1130.79  5131.2 1132.66  5141.9 1135.81  5162.8 1136.19
  5199.8 1142.12  5226.1 1145.31  5231.4 1147.22  5236.7 1146.99  5278.8 1151.57
#Mann= 3 ,-1 , 0
  4804.5     .05       0  4986.6     .05       0  5012.8     .05       0
Bank Sta=4986.6,5012.8
XS Rating Curve= 0 ,0
Exp/Cntr=0.3,0.1

Type RM Length L Ch R = 1 ,18882   ,508,508,508
BEGIN DESCRIPTION:
Mapping XS 541ec96c
END DESCRIPTION:
XS GIS Cut Line= 4
      2788164.94     10223167.73      2788461.81     10223178.15
      2788737.86     10223188.57      2789086.79     10223162.53
#Sta/Elev= 30
  4624.1 1157.81  4664.9 1154.88  4694.9 1154.88  4714.9 1153.08  4774.9 1152.09
  4784.9 1153.56    4845 1149.25    4915 1130.37    4920 1124.15    4935 1121.91
  4955.1 1117.33  5001.9 1115.66  5002.4 1115.16  5028.2 1115.66  5035.1 1117.46
  5045.1 1117.69  5055.1 1119.69  5135.2 1137.28  5175.2 1141.46  5182.8 1141.38
  5187.8 1140.13  5197.4 1141.04  5201.9 1142.84  5235.3 1146.13  5285.5 1147.36
  5315.6 1146.95  5334.2 1145.58  5375.7 1145.79  5445.9 1144.36  5547.3 1149.67
#Mann= 3 ,-1 , 0
  4624.1     .05       0  5001.9     .05       0  5028.2     .05       0
Bank Sta=5001.9,5028.2
XS Rating Curve= 0 ,0
Exp/Cntr=0.3,0.1

Type RM Length L Ch R = 1 ,18374   ,547,547,547
BEGIN DESCRIPTION:
Mapping XS bfd8b8e7
END DESCRIPTION:
XS GIS Cut Line= 3
      2788211.83     10223693.77      2788644.11     10223667.73
      2789200.05     10223678.13
#Sta/Elev= 30
  4716.6 1144.73  4750.5 1145.05  4770.6 1143.67  4790.6 1143.78  4808.2 1142.93
  4816.3  1141.1  4830.7 1139.57  4850.7 1135.68  4878.9 1131.56  4950.9 1117.13
  4957.8 1112.44  4958.3 1111.94  4984.1 1112.44    4991 1113.18    5001 1112.74
  5051.1 1114.25  5081.1 1118.93  5147.9 1124.39  5321.3 1130.77  5361.3 1133.34
  5471.3 1138.31  5491.4 1140.17  5521.3 1141.81  5531.3 1143.72  5541.3 1144.44
  5561.3 1144.75  5571.3 1146.52  5601.3 1149.47  5671.3 1155.02  5705.7 1159.71
#Mann= 7 ,-1 , 0
  4716.6     .05       0  4816.3     .12       0  4878.9     .05       0
  4957.8     .05       0  4984.1     .05       0  5361.3     .12       0
  5491.4     .05       0
Bank Sta=4957.8,4984.1
XS Rating Curve= 0 ,0
Exp/Cntr=0.3,0.1

Type RM Length L Ch R = 1 ,17827   ,327,327,327
BEGIN DESCRIPTION:
SIXMILE CREEK 36.0
END DESCRIPTION:
XS GIS Cut Line= 3
      2788305.66     10223953.09        2788649.       10224195.
      2789030.67     10224228.11
#Sta/Elev= 30
    4580 1134.09  4644.1 1136.37  4673.6 1134.36    4739 1132.68  4831.3 1122.05
    4867 1120.96  4923.6 1116.31  4953.2 1111.03  4959.3 1112.03    4968 1109.76
  4988.7 1109.86  5003.6 1109.15  5004.1 1108.65  5029.9 1109.15  5033.9 1111.42
  5046.9 1113.52  5056.9 1112.12    5077 1112.21    5097 1116.64  5137.2 1120.59
    5152 1120.93  5157.3 1122.53  5227.5 1128.62    5265 1133.56  5270.1 1132.19
  5277.7 1132.28  5297.8 1134.93  5327.9 1136.04    5348 1138.59  5383.1 1139.46
#Mann= 4 ,-1 , 0
    4580     .12       0  4988.7     .05       0  5003.6     .05       0
  5029.9     .05       0
Bank Sta=5003.6,5029.9
XS Rating Curve= 0 ,0
Exp/Cntr=0.3,0.1

Type RM Length L Ch R = 1 ,17500   ,500,500,500
BEGIN DESCRIPTION:
SIXMILE CREEK 35.0
END DESCRIPTION:
XS GIS Cut Line= 3
      2788505.68     10224603.11      2788691.28     10224514.42
      2788955.71     10224303.09
#Sta/Elev= 30
  4794.3 1130.22  4816.5 1129.04  4893.6 1119.43  4905.1 1116.72  4921.2 1115.25
  4938.4  1114.5  4967.2 1110.54  4982.7 1109.42  5030.5 1108.76    5031 1108.26
  5062.1 1108.76  5068.7  1113.3  5075.1 1113.54  5082.4  1111.8  5095.9 1112.47
  5110.3 1111.81  5124.7 1114.39  5146.5 1114.03  5174.4 1116.36  5188.8 1119.42
  5196.8 1122.21  5210.5 1124.12    5232 1125.45  5238.4 1126.94  5246.4 1126.33
  5281.6 1128.11  5302.4 1130.18  5310.5 1132.32  5316.9 1132.17  5338.5 1134.91
#Mann= 4 ,-1 , 0
  4794.3     .05       0  4921.2     .12       0  5030.5     .07       0
  5062.1     .05       0
Bank Sta=5030.5,5062.1
XS Rating Curve= 0 ,0
Exp/Cntr=0.3,0.1
